HEC-RAS study BAYOU CREEK.prj: BAYOU CREEK Base Level Engineering

--- BAYOU CREEK.g01 (geometry) --- (continued)

Type RM Length L Ch R = 1 ,42053   ,694,694,694
BEGIN DESCRIPTION:
BAYOU CREEK 63.0
END DESCRIPTION:
XS GIS Cut Line= 3
      2364086.45     13221471.86      2363686.41     13221421.85
      2362986.37     13221321.85
#Sta/Elev= 30
  4547.1  125.21  4596.2  125.35  4624.6  125.07  4727.2  125.12  4790.9  121.96
  4858.2  116.74  4888.5  115.42  4908.6  112.51  4938.9  109.75  4979.2  101.96
  4986.3   94.89  4989.1   94.39  4999.4   95.69  5009.5   102.2  5022.8  101.43
  5029.7  102.64  5070.1  104.44  5110.6  103.31    5151  103.88    5252  104.41
  5292.4  105.08  5300.6  106.04  5305.7  105.48  5504.5   117.1  5565.1  119.87
  5583.5  119.99  5588.5  118.73  5615.6  119.28  5625.7  120.77  5657.4  122.25
#Mann= 8 ,-1 , 0
  4547.1     .05       0  4596.2      .1       0  4624.6     .16       0
  4727.2      .1       0  4908.6     .12       0  4999.4     .12       0
    5151     .16       0  5504.5      .1       0
Bank Sta=4979.2,5009.5
XS Rating Curve= 0 ,0
Exp/Cntr=0.3,0.1

Type RM Length L Ch R = 1 ,41359   ,658,658,658
BEGIN DESCRIPTION:
BAYOU CREEK 62.0
END DESCRIPTION:
XS GIS Cut Line= 4
      2364042.05     13221076.95      2363822.65      13220799.8
      2363268.36     13220770.93      2363108.01     13220862.56
#Sta/Elev= 30
  4250.9  124.38  4317.7  123.97  4353.1   122.6  4381.8  122.26  4518.1  116.27
  4524.5  116.66  4629.3  111.58  4749.5  108.34  4799.6  105.07  4859.7  102.75
  4969.8  102.12  4979.8  100.49  4989.8   93.04  4999.6   91.28  5002.8   91.78
  5009.9   99.55  5018.5   99.36  5029.9  100.72  5039.9  101.57    5100  106.71
    5130  111.17  5179.4  110.33  5222.6  111.76  5252.3  111.11  5260.1  110.66
  5287.4  111.98  5297.5  111.43  5303.2  112.28  5319.1     112  5344.1  113.18
#Mann= 6 ,-1 , 0
  4250.9     .05       0  4353.1      .1       0  5009.9     .07       0
  5018.5      .1       0  5029.9     .16       0  5252.3      .1       0
Bank Sta=4969.8,5039.9
XS Rating Curve= 0 ,0
Exp/Cntr=0.3,0.1

Type RM Length L Ch R = 1 ,40701   ,579,579,579
BEGIN DESCRIPTION:
BAYOU CREEK 61.0
END DESCRIPTION:
XS GIS Cut Line= 3
       2364261.9     13221301.64      2363923.34     13220671.41
      2363512.29     13219755.64
#Sta/Elev= 30
  3856.7  123.98  3997.8  123.21  4100.5  124.47  4145.5  123.79  4151.2  124.58
  4189.4  123.31    4195  124.16  4670.8  104.16  4740.3  103.58  4838.5  100.33
  4905.9  101.15  4927.9   98.94  4949.8   99.83  4971.7   99.34  4988.5   97.78
  4993.9   94.01  5004.3   91.25  5017.1   95.02  5026.5  100.31    5058  106.04
  5086.6  108.45  5103.2  111.31  5147.1  114.86  5161.6  115.11    5169  116.46
  5306.1  123.89    5443  126.69    5497  126.23  5502.5  126.88  5575.9  125.65
#Mann= 11 ,-1 , 0
  3777.7     .16       0  3862.6      .1       0  4392.3     .05       0
  4577.1      .1       0    4772     .12       0  4993.8     .07       0
  4999.8     .12       0    5033      .1       0  5041.8     .12       0
  5153.9     .16       0  5312.6      .1       0
Bank Sta=4971.7,5026.5
XS Rating Curve= 0 ,0
Exp/Cntr=0.3,0.1

Type RM Length L Ch R = 1 ,40122   ,818,818,818
BEGIN DESCRIPTION:
BAYOU CREEK 60.0
END DESCRIPTION:
XS GIS Cut Line= 3
      2364652.52     13221166.24      2364381.67     13220192.24
      2363721.49      13219703.6
#Sta/Elev= 30
  3887.9  124.84    4126  123.91  4177.9  122.73  4302.7  118.42  4437.4  115.27
  4631.5  105.77  4818.3     100  4823.5   98.83  4948.6   97.85  4969.5   99.88
  4977.9   98.95  4984.1   93.48  4990.9   90.44  4998.5   89.04  5013.3   91.18
  5019.6   96.19    5028   98.51  5040.6   99.41  5090.5   98.65  5140.6  102.36
  5177.5   102.1  5305.5  104.19  5313.9  105.24    5341   105.6  5470.4  111.15
  5491.3  111.11  5570.6  114.76  5591.5   114.3  5599.9  115.33  5720.2  117.89
#Mann= 11 ,-1 , 0
  3780.8      .1       0    4428     .05       0  4531.3      .1       0
  4634.7     .12       0  4714.4      .1       0  4845.9     .12       0
    5000     .07       0    5006     .12       0  5129.4      .1       0
  5400.8     .16       0  5579.7      .1       0
Bank Sta=4969.5,5040.6
XS Rating Curve= 0 ,0
Exp/Cntr=0.3,0.1

Type RM Length L Ch R = 1 ,39304   ,463,463,463
BEGIN DESCRIPTION:
Mapping XS 9f7edd60
END DESCRIPTION:
XS GIS Cut Line= 3
      2364876.46     13220239.09      2364787.92     13219843.28
      2363803.53     13219098.48
#Sta/Elev= 30
  4050.4  110.64  4067.8  111.29  4246.5  107.36  4251.6   108.3  4430.4  108.87
  4504.1  111.07  4560.3  105.55  4589.4   99.08    4604   98.27  4610.3   99.33
  4639.4    95.9    4682   96.12  4689.3   94.63  4703.9   94.46  4753.8   97.83
  4924.5   99.48  4974.4   95.92  4982.7    95.6  4992.5   87.73  4995.2   87.23
  5009.8   90.43  5018.1   96.81  5059.7    96.8    5068   98.38  5124.2   98.45
  5182.4  100.88  5246.3  105.31  5338.5  115.19  5367.6  117.01  5690.4  125.97
#Mann= 12 ,-1 , 0
    4033     .05       0  4074.1      .1       0  4430.9     .16       0
  4655.8      .1       0  4894.3     .16       0  4920.7     .12       0
  4994.4     .07       0  5000.4     .12       0  5378.4     .16       0
  5431.7      .1       0  5481.3     .16       0  5617.1      .1       0
Bank Sta=4974.4,5018.1
XS Rating Curve= 0 ,0
Exp/Cntr=0.3,0.1

Type RM Length L Ch R = 1 ,38841   ,574,574,574
BEGIN DESCRIPTION:
BAYOU CREEK 59.0
END DESCRIPTION:
XS GIS Cut Line= 2
      2364912.95     13219447.47       2364059.7     13218771.11
#Sta/Elev= 30
    4524  110.06  4563.9   111.6  4677.7  108.15  4820.3   99.75  4905.2   96.14
  4977.3   94.89  4980.7    86.2  4983.5    85.7  4990.1   87.11  5004.5   86.88
  5012.6   94.19  5041.1   96.29  5062.3   95.83  5068.6   94.45  5076.7   95.83
  5132.7   96.84  5140.8   98.35  5147.2    97.8  5155.2   99.72    5176  100.12
  5182.4  101.98  5196.8   102.1  5204.9  103.69  5246.5  106.57  5382.7  112.31
  5403.6  112.23    5418  113.63  5446.8  114.47  5560.6  115.28  5612.8  117.34
#Mann= 6 ,-1 , 0
  4518.3      .1       0  4697.9     .16       0  5000.6     .07       0
  5006.6     .16       0  5016.2     .12       0  5154.8      .1       0
Bank Sta=4977.3,5012.6
XS Rating Curve= 0 ,0
Exp/Cntr=0.3,0.1

Type RM Length L Ch R = 1 ,38267   ,390,390,390
BEGIN DESCRIPTION:
BAYOU CREEK 58.0
END DESCRIPTION:
XS GIS Cut Line= 3
      2364936.41     13219371.81      2364936.41     13218721.85
      2364586.39     13218471.84
#Sta/Elev= 30
  4397.3  108.73  4492.3  105.93  4572.3  100.69  4642.3   98.27  4762.3    98.2
  4802.3   96.52  4892.3   95.84  4942.3   94.16  4952.3   94.59  4982.3   93.82
  4992.3   88.58    5002   86.02  5005.3   86.52  5032.3      96  5042.3   98.37
  5047.3   98.37  5049.5  100.79  5064.3  100.95  5070.4  102.34  5085.2  103.78
  5093.8  103.14  5099.9  103.75  5120.8  103.49  5150.3     105  5215.4  105.09
  5221.6  104.43    5230  105.15  5307.6  104.87  5378.9  106.17  5477.4  109.74
#Mann= 7 ,-1 , 0
    4325      .1       0  4721.7     .16       0  4732.8     .12       0
  4997.4     .16       0  5000.3     .07       0  5006.3     .16       0
  5271.9     .05       0
Bank Sta=4982.3,5032.3
XS Rating Curve= 0 ,0
Exp/Cntr=0.3,0.1

Type RM Length L Ch R = 1 ,37877   ,331,331,331
BEGIN DESCRIPTION:
Mapping XS c2f3b900
END DESCRIPTION:
XS GIS Cut Line= 3
      2366126.47     13218900.57      2365366.05     13218733.91
      2364709.83     13218265.18
#Sta/Elev= 30
  4158.9  115.54  4403.3  115.54  4572.8  109.29  4679.7  109.54  4700.2   107.2
  4730.9  109.03  4751.4   107.6  4758.3   100.9  4763.4  100.78  4782.1   95.93
  4807.3    95.9  4833.3   98.44  4884.5   94.55    4900   84.84  4915.2   86.61
  4925.4   93.24  4962.1   94.07  4970.7   93.17  4984.5   86.58  4997.5    83.9
  5006.3   84.66  5012.5   90.84  5027.2   94.23  5048.1   95.17  5083.7   92.82
  5119.7   95.58  5148.9    95.1    5300   99.56    5493  101.85  5743.8  110.05
#Mann= 12 ,-1 , 0
  4029.9      .1       0  4344.7     .05       0  4445.5     .16       0
    4505     .05       0  4545.3     .16       0  4560.3     .12       0
  4907.6     .16       0  5001.1     .07       0  5007.1     .16       0
  5061.9     .12       0    5206     .16       0  5452.5     .05       0
Bank Sta=4962.1,5027.2
XS Rating Curve= 0 ,0
Exp/Cntr=0.3,0.1

Type RM Length L Ch R = 1 ,37546   ,490,490,490
BEGIN DESCRIPTION:
BAYOU CREEK 57.0
END DESCRIPTION:
XS GIS Cut Line= 3
      2366157.68     13218791.18      2365483.02     13218453.06
      2364697.77     13217921.66
#Sta/Elev= 30
  4142.5   113.9  4250.7  111.13    4502  109.39  4630.5  111.38  4658.5  103.65
  4668.2  103.53  4675.2  105.34  4735.3   99.62  4757.7  101.37  4770.2   96.63
    4780   96.47  4802.4   97.38  4809.3  101.09  4814.9   98.64  4891.7   98.94
  4955.4   96.55  4976.3   92.72  4985.3   85.17  4997.1   83.65  4999.9   83.15
  5003.1   83.65  5021.2   87.87  5027.3   85.89  5036.2   91.29  5057.2   92.15
  5072.1   93.22  5108.1   94.01  5251.9   99.24  5446.6  100.17  5845.3  118.93
#Mann= 10 ,-1 , 0
  4142.5     .05       0  4250.7      .1       0  4668.2     .05       0
  4735.3     .08       0  4891.7     .16       0  4997.1     .07       0
  5003.1     .16       0  5072.1     .12       0  5108.1     .16       0
  5251.9     .05       0
Bank Sta=4976.3,5057.2
XS Rating Curve= 0 ,0
Exp/Cntr=0.3,0.1

Type RM Length L Ch R = 1 ,37056   ,410,410,410
BEGIN DESCRIPTION:
BAYOU CREEK 56.0
END DESCRIPTION:
XS GIS Cut Line= 3
      2366277.46     13218249.51      2365855.63     13218021.85
      2364871.99     13217760.14
#Sta/Elev= 30
  4180.3  116.36  4212.9  115.11  4293.6  113.55  4404.3  113.53  4491.8  110.58
  4529.9  110.54  4535.6  109.23  4617.5  105.73  4896.8   91.99  4947.2   93.96
  4957.6   93.12  4978.3   87.92  4988.6   83.13    4996   82.77  4998.7   82.27
  5006.9   85.65  5012.1   86.87  5019.7    91.2    5030   91.75  5071.4   92.86
  5092.4   95.47  5112.8   95.91  5143.8   99.43  5162.3   99.14  5207.6  101.93
  5257.7  104.92  5443.9  111.59  5537.1  113.71  5588.3  113.53  5677.5  116.12
#Mann= 10 ,-1 , 0
  4180.3     .05       0  4212.9      .1       0  4617.5     .16       0
  4988.6     .07       0    4996     .16       0  5006.9     .12       0
  5112.8      .1       0  5162.3     .05       0  5207.6      .1       0
  5588.3     .05       0
Bank Sta=4957.6,5030
XS Rating Curve= 0 ,0
Exp/Cntr=0.3,0.1

Type RM Length L Ch R = 1 ,36646   ,493,493,493
BEGIN DESCRIPTION:
BAYOU CREEK 55.0
END DESCRIPTION:
XS GIS Cut Line= 3
       2366336.4     13217621.85      2365786.41     13217571.85
      2365086.45     13217621.85
#Sta/Elev= 30
  4380.1  116.75  4418.9  116.22  4469.1  113.96  4509.3  112.29  4589.6  108.28
  4609.7  107.75  4700.1  102.19  4823.8   93.94  4880.8   90.58  4909.4   90.12
  4951.1   91.35  4971.1   90.12  4981.2   85.33  4991.2   83.17    5001    82.6
  5011.2   84.18  5021.3   90.84  5031.3   92.72  5041.3   91.75  5074.6   91.41
  5091.5   92.04  5101.5   93.59  5131.6   94.47  5151.6   96.25  5209.9   98.99
  5402.2  106.88  5452.4  108.22  5490.6  109.85  5502.5   111.1  5634.1  112.37
#Mann= 11 ,-1 , 0
  4380.1     .05       0  4418.9     .16       0  4469.1      .1       0
  4509.3     .16       0  4589.6      .1       0  4700.1     .12       0
  4823.8      .1       0  4909.4     .12       0    5001     .07       0
  5011.2     .12       0  5209.9     .05       0
Bank Sta=4951.1,5031.3
XS Rating Curve= 0 ,0
Exp/Cntr=0.3,0.1

Type RM Length L Ch R = 1 ,36153   ,514,514,514
BEGIN DESCRIPTION:
BAYOU CREEK 54.0
END DESCRIPTION:
XS GIS Cut Line= 3
      2366386.44     13217321.87      2366036.41     13217121.85
      2365236.45     13217421.84
#Sta/Elev= 30
  4503.1  108.67  4542.7  108.58  4580.1  106.84    4732   97.32  4843.6   91.95
  4865.2   91.49  4893.2   87.39  4933.1   89.45  4958.1   92.44  4963.4   92.35
  4968.9   91.95  4988.3   81.26  4993.7   81.28  5000.7   80.03    5004   80.53
  5011.6   87.82  5018.6   91.57  5023.9   90.34    5033   91.57  5054.4   90.25
    5065   90.69  5073.8   92.27  5086.4   92.55  5164.5   91.12  5219.7   91.54
  5289.3   94.81  5374.8   96.01    5567   96.65  5671.8   98.98  5760.6  102.41
#Mann= 12 ,-1 , 0
  4503.1     .05       0  4580.1      .1       0    4732     .16       0
  4843.6      .1       0  4958.1     .16       0  4963.4     .12       0
  4988.3     .07       0  4993.7     .12       0    5004     .16       0
    5065     .12       0  5164.5     .16       0  5374.8     .05       0
Bank Sta=4963.4,5018.6
XS Rating Curve= 0 ,0
Exp/Cntr=0.3,0.1

Type RM Length L Ch R = 1 ,35639   ,720,720,720
BEGIN DESCRIPTION:
BAYOU CREEK 53.0
END DESCRIPTION:
XS GIS Cut Line= 3
      2366688.94      13216728.7      2365360.84     13216577.66
      2364845.22     13216957.86
#Sta/Elev= 30
  4353.4   117.5    4405  116.99  4656.6  111.95  4680.6  113.96  4686.8  111.18
    4727  108.85  4827.7  100.61  4918.2   89.84  4978.6   90.09  4988.7   87.76
  4995.8   81.19  4998.5   80.69  5001.8   81.19  5028.7   85.64    5039   90.66
  5049.1   92.32  5129.6   89.51  5159.8   90.43    5200   91.34    5502   92.67
  5612.7   97.27  5706.4  100.39  5805.8  101.06  5855.5  100.68  5934.6  100.41
  5949.3   96.32  5955.5   98.74  5963.9   95.17  5984.8  100.72  6330.7  110.23
#Mann= 13 ,-1 , 0
  4353.4     .05       0    4405     .16       0    4727      .1       0
  4827.7     .12       0  4995.8     .07       0  5001.8     .12       0
  5159.8     .16       0    5200     .12       0    5502      .1       0
  5612.7     .05       0  5706.4      .1       0  5805.8     .05       0
  5855.5      .1       0
Bank Sta=4978.6,5049.1
XS Rating Curve= 0 ,0
Exp/Cntr=0.3,0.1

Type RM Length L Ch R = 1 ,34919   ,585,585,585
BEGIN DESCRIPTION:
BAYOU CREEK 52.0
END DESCRIPTION:
XS GIS Cut Line= 3
      2366436.41     13216121.85      2366036.41     13216071.85
      2365236.38     13216121.86
#Sta/Elev= 30
  4346.3  111.67  4355.1  111.48  4556.6  111.77  4637.2  108.47  4749.4  102.99
  4818.2   97.58  4868.3   91.91  4906.6   91.42  4918.4   90.12  4948.5   90.66
  4958.5   90.38  4978.5   87.54  4988.6    82.6  4998.6   79.98  5005.6   79.98
  5008.4   79.48  5028.6   84.55  5038.7   90.23  5048.7   90.45  5058.7   83.18
  5066.9   81.41  5071.9   84.07  5098.8    82.3  5128.8   89.81  5148.9   89.93
  5299.2   89.58  5369.3   91.14  5469.5   97.78  5539.6  101.85    5551  102.13
#Mann= 10 ,-1 , 0
  4346.3     .05       0  4355.1     .05       0  4637.2      .1       0
  4978.5     .12       0  5005.6     .07       0  5008.4     .12       0
  5148.9     .16       0  5369.3      .1       0  5469.5     .12       0
  5539.6      .1       0
Bank Sta=4948.5,5048.7
XS Rating Curve= 0 ,0
Exp/Cntr=0.3,0.1

Type RM Length L Ch R = 1 ,34334   ,459,459,459
BEGIN DESCRIPTION:
BAYOU CREEK 51.0
END DESCRIPTION:
XS GIS Cut Line= 3
      2366392.09     13215879.74      2365819.17     13215530.78
      2365162.91     13215634.95
#Sta/Elev= 30
  4045.7  106.46  4051.2  106.46  4058.8  108.04  4196.3  109.78  4248.6  108.21
  4291.2   104.8  4349.3  102.06  4378.7   99.58  4495.8   92.95  4502.3   94.19
  4508.2   92.74  4539.1   92.46  4560.4   90.93  4768.6   88.85    4880   88.92
  4971.1   88.37  4977.4    85.5  4982.4   81.55  5001.2   79.17  5004.5   79.67
  5011.6   82.94  5021.8   87.56  5044.7   86.78  5072.4   87.44  5193.9   95.04
  5254.6   96.48  5293.8   95.21  5298.8   96.63  5335.6   96.12    5381   98.03
#Mann= 6 ,-1 , 0
  4045.7     .05       0  4196.3      .1       0    4880     .12       0
  5011.6     .12       0  5072.4      .1       0  5193.9     .16       0
Bank Sta=4971.1,5021.8
XS Rating Curve= 0 ,0
Exp/Cntr=0.3,0.1

Type RM Length L Ch R = 1 ,33875   ,564,564,564
BEGIN DESCRIPTION:
BAYOU CREEK 50.0
END DESCRIPTION:
XS GIS Cut Line= 3
      2366336.42     13215771.86      2365636.41     13215171.85
      2365286.39     13214971.84
#Sta/Elev= 30
  4030.4  107.97  4054.8  108.58  4096.5  108.43  4104.2  109.52  4358.8   93.33
    4437   90.19  4529.2   89.33  4628.8   89.22  4792.4   87.49  4827.5   88.85
  4862.6   86.36  4952.4   89.04  4954.5   88.86  4970.3   87.96  4994.7   78.73
  4997.4   78.23  5000.7   78.73  5007.8   81.83  5013.5   82.64    5020   86.51
  5050.9   88.83  5056.7   88.93  5094.1   99.19  5100.6  101.81    5110  102.63
  5115.7  100.84  5123.6  104.18  5146.7  106.73  5212.2  107.45  5355.5  109.06
#Mann= 9 ,-1 , 0
  4030.4     .05       0  4054.8      .1       0  4529.2     .12       0
  4628.8      .1       0  4952.4     .12       0  4994.7     .07       0
  5000.7     .12       0  5094.1      .1       0  5212.2     .05       0
Bank Sta=4954.5,5050.9
XS Rating Curve= 0 ,0
Exp/Cntr=0.3,0.1

Type RM Length L Ch R = 1 ,33311   ,497,497,497
BEGIN DESCRIPTION:
BAYOU CREEK 49.0
END DESCRIPTION:
XS GIS Cut Line= 4
      2367522.32      13214853.7      2366715.01     13214937.03
      2366381.67     13215108.91      2365341.39      13214713.6
#Sta/Elev= 30
  3455.9  116.43  3902.9  106.37  4083.8   106.1  4451.3   93.25  4534.4   88.03
  4545.7    84.8  4584.3   89.27  4678.9    87.2  4717.5   90.73  4722.8   88.28
  4764.4   90.38  4839.3   85.02  4967.2   87.43  4997.1   76.71  5042.6    87.2
  5160.3   87.62  5267.2   97.72  5406.3  103.58  5482.7  104.81  5502.1   99.79
  5507.4  104.75    5524  104.82  5532.2  100.66  5537.6  102.73  5545.4   99.58
  5562.3   98.35  5609.6  102.26  5622.6  107.76  5684.4  107.71  5755.4  112.07
#Mann= 10 ,-1 , 0
  3165.3     .05       0  3574.9      .1       0  3889.9     .05       0
  4039.9     .12       0  4222.1      .1       0  4445.4     .12       0
  4950.1     .07       0  5035.1     .12       0  5041.6      .1       0
  5353.1     .05       0
#XS Ineff= 2 , 0
         4284.09   95.91
Permanent Ineff=
       F       F
Bank Sta=4967.2,5042.6
XS Rating Curve= 0 ,0
Exp/Cntr=0.3,0.1

Type RM Length L Ch R = 1 ,32814   ,711,711,711
BEGIN DESCRIPTION:
BAYOU CREEK 48.0
END DESCRIPTION:
XS GIS Cut Line= 3
      2367563.94     13214681.82      2366511.88     13214650.57
       2365491.9     13214452.82
#Sta/Elev= 30
  3801.5  106.39    4135  101.59  4147.9  103.69  4177.9  101.71  4237.9  102.29
    4368   96.13    4518   96.37  4578.1   94.56  4698.1   94.18  4878.6   87.09
  4896.9   87.67    4902   89.17  4939.8   87.35  4980.5   85.82  4987.7   75.49
  4990.4   74.99  5005.4   76.64  5011.1    79.1  5041.6   80.41  5062.3   86.86
    5225   85.89  5372.7   89.54  5377.8   90.79  5449.1   92.89    5500   97.58
  5601.9   99.83  5631.4  104.11    5663  103.67  5791.7   109.3    5893  111.02
#Mann= 10 ,-1 , 0
  3772.7     .05       0  4425.8      .1       0    4676     .12       0
  4757.1     .05       0  4971.3     .12       0  4990.8     .07       0
  4996.8     .12       0  5120.9      .1       0  5490.9     .16       0
  5603.9     .05       0
Bank Sta=4939.8,5062.3
XS Rating Curve= 0 ,0
Exp/Cntr=0.3,0.1

Type RM Length L Ch R = 1 ,32103   ,363,363,363
BEGIN DESCRIPTION:
BAYOU CREEK 47.0
END DESCRIPTION:
XS GIS Cut Line= 3
      2367322.68     13214216.89      2366371.17     13214233.28
      2365605.37     13214126.18
#Sta/Elev= 30
  3917.7  112.48  4112.7  110.52  4206.8  106.85  4402.7   96.35  4572.8   90.29
  4652.8   88.76  4722.8   88.88  4852.8   83.23  4878.8   85.16  4913.2    84.6
  4973.8   83.34  4983.9   79.36    4991   74.41  4993.8   73.91  5004.1   75.24
  5014.2   80.12  5021.6   85.32  5084.9    85.4  5125.3   86.57  5155.6   89.66
  5169.6   89.58  5296.9   97.43    5307   98.79  5367.6  101.01  5428.2  104.85
  5526.8  107.41  5559.5  107.44  5569.5  108.53  5579.6  107.69  5642.6  106.96
#Mann= 8 ,-1 , 0
       0     .05       0653.6032      .1       0911.0833     .12       0
1000.084     .05       01256.902     .12       01286.535     .07       0
1316.168     .12       0 1474.21      .1       0
Bank Sta=4913.2,5021.6
XS Rating Curve= 0 ,0
Exp/Cntr=0.3,0.1

Type RM Length L Ch R = 1 ,31740   ,511,511,511
BEGIN DESCRIPTION:
BAYOU CREEK 46.0
END DESCRIPTION:
XS GIS Cut Line= 3
      2367176.85     13213661.32      2366624.73     13213859.25
      2365836.58     13214025.91
#Sta/Elev= 30
    4201  112.24  4253.2  111.93  4316.4  110.39  4383.2  108.59  4495.6  103.13
  4593.1   96.81    4625   93.96  4761.7   86.87  4844.6   85.65  4917.3   86.53
    4944   84.12  4968.4   83.56  4988.6   80.67  4993.7   81.37  4996.1    73.2
  4998.9    72.7  5009.3   75.28  5019.6   82.31  5038.3   81.87  5070.7   82.84
  5080.9   84.54  5093.2    84.7  5111.5   84.73  5162.7   85.02  5172.9   83.75
  5187.5   83.78  5193.3   84.53  5305.7   87.22  5381.3   90.55  5593.1  102.81
#Mann= 6 ,-1 , 0
    4201     .05       0  4253.2      .1       0  4316.4     .12       0
  4993.7     .07       0  4998.9     .12       0  5111.5     .05       0
Bank Sta=4917.3,5093.2
XS Rating Curve= 0 ,0
Exp/Cntr=0.3,0.1

Type RM Length L Ch R = 1 ,31229   ,649,649,649
BEGIN DESCRIPTION:
BAYOU CREEK 45.0
END DESCRIPTION:
XS GIS Cut Line= 3
      2367159.49     13213501.62      2366340.01     13213383.56
      2365842.32     13213062.14
#Sta/Elev= 30
  4282.3   109.1  4364.7  108.76    4375  108.57  4577.1  101.28  4637.7    99.1
  4697.4   98.43  4809.5   92.88  4870.1   88.47  4930.7   83.54    4961   81.81
  4971.1   82.48  4979.1   78.67  4984.1   78.56  4988.3   73.73  4991.1   73.23
  5001.4   73.83  5011.5   80.01  5021.6   82.29  5049.5   83.49  5082.2   82.65
  5152.4   83.14  5167.6   81.71  5240.2    84.6  5276.5   84.75  5349.1   84.59
  5421.6   88.06  5442.8   90.01  5542.4   95.74  5645.3  100.39  5702.7     102
#Mann= 11 ,-1 , 0
  4282.3     .05       0  4364.7     .05       0    4375     .16       0
  4577.1      .1       0  4870.1     .05       0  4971.1     .12       0
  4991.1     .07       0  5001.4     .12       0  5167.6     .05       0
  5276.5     .12       0  5645.3      .1       0
Bank Sta=4930.7,5049.5
XS Rating Curve= 0 ,0
Exp/Cntr=0.3,0.1

Type RM Length L Ch R = 1 ,30580   ,463,463,463
BEGIN DESCRIPTION:
BAYOU CREEK 44.0
END DESCRIPTION:
XS GIS Cut Line= 3
      2367218.47     13213262.03      2366863.16     13212794.23
      2365873.99     13212709.91
#Sta/Elev= 30
  4018.6  103.29  4108.7  101.52  4158.7  100.24  4200.9   100.7  4208.6   99.61
  4287.6   98.07  4293.9   98.69  4372.9   95.46  4464.6   93.32  4472.7   92.05
    4606   91.13  4711.9   86.79  4832.3   83.83  4922.6   81.26  4962.8    82.8
  4972.8   82.78  4987.5   80.81  4992.9   73.69  4999.9   73.63  5002.7   73.13
    5023   74.86    5033    82.1  5043.1   82.56  5073.2   82.28  5133.4   81.35
  5173.5   84.77  5220.7   88.95  5324.1   94.66  5453.8   98.59  5598.8  100.92
#Mann= 7 ,-1 , 0
  4018.6     .05       0  4108.7      .1       0  4832.3     .12       0
  4999.9     .07       0  5002.7     .12       0  5073.2     .05       0
  5173.5      .1       0
Bank Sta=4962.8,5043.1
XS Rating Curve= 0 ,0
Exp/Cntr=0.3,0.1

Type RM Length L Ch R = 1 ,30117   ,359,359,359
BEGIN DESCRIPTION:
BAYOU CREEK 43.0
END DESCRIPTION:
XS GIS Cut Line= 3
      2366986.45     13212221.85      2366586.41     13212221.85
      2366136.42     13212621.84
#Sta/Elev= 30
  4471.5  102.04  4610.2   99.53  4690.2   97.26  4700.2   96.03  4800.2   90.86
  4810.2   89.19  4868.4   84.42  4888.2   84.07  4895.7   82.66  4930.9   80.23
    4966   80.11  4980.2   82.18  4987.7    74.3  5001.9   72.76  5005.6   72.29
  5008.4   71.79  5011.6   72.29  5016.2   74.74  5022.9   75.28  5030.3    79.5
  5065.5   83.07  5086.4   83.37  5129.1   81.45  5206.8      81  5228.6   83.23
  5263.7    84.6    5349   87.74  5355.7   88.96  5412.5   89.36  5473.6   91.98
#Mann= 8 ,-1 , 0
  4471.5     .05       0  4610.2     .05       0  4700.2      .1       0
  4930.9     .12       0  5001.9     .07       0  5005.6     .12       0
  5129.1     .05       0  5263.7      .1       0
Bank Sta=4980.2,5065.5
XS Rating Curve= 0 ,0
Exp/Cntr=0.3,0.1

Type RM Length L Ch R = 1 ,29758   ,844,844,844
BEGIN DESCRIPTION:
BAYOU CREEK 42.0
END DESCRIPTION:
XS GIS Cut Line= 2
      2367048.31     13211921.76      2365708.09     13212001.61
#Sta/Elev= 30
  4374.5   99.87  4445.2   99.61  4515.3   97.09  4542.3   95.98  4716.6   95.67
  4755.8   94.87  4795.8   93.66  4845.9   90.33    4866   88.22    4896   84.77
  4936.1   81.47  4956.1   80.26  4976.2   81.74  4986.2   79.72  4996.2   72.88
  5006.2   72.09    5016   71.55  5019.2   72.05  5026.2   77.18    5050   82.47
  5076.3   82.55  5156.5   79.88  5246.6   84.24  5356.8   81.11    5437   80.98
  5497.1   82.63  5547.2   85.17  5677.4   92.25  5697.4   93.54  5717.1   94.98
#Mann= 11 ,-1 , 0
  4374.5     .05       0  4515.3      .1       0    4866     .12       0
  5006.2     .12       0  5156.5     .05       0  5246.6     .12       0
  5356.8      .1       0    5437     .12       0  5547.2      .1       0
  5677.4     .12       0  5697.4      .1       0
Bank Sta=4936.1,5050
XS Rating Curve= 0 ,0
Exp/Cntr=0.3,0.1

Type RM Length L Ch R = 1 ,28914   ,1093,1093,1093
BEGIN DESCRIPTION:
BAYOU CREEK 41.0
END DESCRIPTION:
XS GIS Cut Line= 3
      2367072.66     13211741.21      2366683.76     13211487.73
      2365936.39     13211021.84
#Sta/Elev= 30
  3968.6   97.43    4070   97.75    4249   89.04    4321   86.77  4460.2   88.23
  4633.7   82.86  4764.6   80.64    4859    80.9  4880.3      82  4953.4   81.97
  4959.3   81.67  4968.8   77.32  4974.7   77.23    4982   72.72    4990   70.93
  4995.9   71.23  5002.3    70.7  5005.1    70.2  5008.3    70.7  5017.3   79.25
  5026.6   78.65  5053.7   82.45  5063.2   84.01  5084.4   83.97  5111.6    88.3
  5135.2   89.07  5157.6   91.46  5205.9    93.1  5242.5   94.53  5313.5   96.37
#Mann= 8 ,-1 , 0
  3968.6     .05       0    4070      .1       0    4859     .12       0
  4995.9     .07       0  5002.3     .12       0  5063.2     .05       0
  5205.9      .1       0  5242.5     .05       0
Bank Sta=4953.4,5053.7
XS Rating Curve= 0 ,0
Exp/Cntr=0.3,0.1

Type RM Length L Ch R = 1 ,27821   ,531,531,531
BEGIN DESCRIPTION:
BAYOU CREEK 40.0
END DESCRIPTION:
XS GIS Cut Line= 3
      2367149.04     13211727.32      2367018.83     13211076.27
      2366742.76     13210633.52
#Sta/Elev= 30
  4208.2   93.34  4412.6   94.26  4497.3    91.1  4594.2   85.99    4637   86.01
  4645.2    84.1  4667.6   82.54  4701.3    81.8  4747.2   78.68    4790   77.16
  4830.8   78.02  4840.9   75.87  4854.3   75.36  4861.3   77.45  4880.5   78.15
  4901.7   78.73  4938.3   76.86  4965.7   78.96  4980.8   78.84  4996.1   69.28
  5011.2   68.26  5024.7   71.95  5032.7      78  5048.1   78.52  5075.2   77.89
  5111.8   79.27  5177.9   85.26  5242.7   89.72  5307.5   91.42  5393.9   90.75
#Mann= 5 ,-1 , 0
  4131.3      .1       0  4831.9     .12       0  4993.6     .07       0
  4999.6     .12       0  5144.7      .1       0
Bank Sta=4965.7,5048.1
XS Rating Curve= 0 ,0
Exp/Cntr=0.3,0.1

Type RM Length L Ch R = 1 ,27290   ,563,563,563
BEGIN DESCRIPTION:
BAYOU CREEK 39.0
END DESCRIPTION:
XS GIS Cut Line= 3
      2367878.19     13211018.97      2367149.04     13210576.27
       2366784.5     13210607.51
#Sta/Elev= 30
  4459.1  105.97  4496.3   104.6  4527.3  104.86  4723.1   96.05  4728.9   94.43
  4765.8      91  4839.4   85.93  4845.7    84.4  4876.2   82.77    4913   78.76
  4940.2   76.88  4971.2    77.1    4977    72.1  4986.1   69.07  4998.1   67.45
    5008   69.67  5013.8   74.17  5021.2   76.53  5029.3   76.99  5050.7   78.16
  5056.5      77  5196.7   77.97  5225.1    80.9  5255.2   79.03  5333.5   78.93
  5403.8   81.13  5413.8   84.04  5433.9   81.74  5564.4   86.85    5678   89.51
#Mann= 6 ,-1 , 0
  4415.2      .1       0  4936.6     .12       0  4999.7     .07       0
  5005.7     .12       0  5168.9     .05       0    5280      .1       0
Bank Sta=4971.2,5029.3
XS Rating Curve= 0 ,0
Exp/Cntr=0.3,0.1

Type RM Length L Ch R = 1 ,26727   ,296,296,296
BEGIN DESCRIPTION:
BAYOU CREEK 38.0
END DESCRIPTION:
XS GIS Cut Line= 3
       2368336.5     13210420.01      2367487.58     13210242.93
      2366722.36      13210586.5
#Sta/Elev= 30
  4394.6   116.2  4436.9  115.51  4454.6   115.8    4537  112.21  4658.9  105.97
    4710  102.43    4802    95.7  4812.2   92.86    4853   86.46  4876.9   85.52
  4914.3   81.61  4921.9   78.49    4945   76.94  4955.2   76.49  4965.4   72.09
  4971.9   65.97  4985.6   64.82    4996    65.7  5016.5   70.75  5021.9   76.08
    5027   76.66  5047.1   76.08  5216.9   76.42  5355.8   79.35  5575.3   77.05
  5689.1   78.25  5794.8   81.62  5930.3    86.8  6042.9   89.36  6100.6   89.08
#Mann= 13 ,-1 , 0
  4394.6     .05       0  4436.9      .1       0  4454.6     .16       0
    4537      .1       0  4658.9     .16       0    4710      .1       0
  4955.2     .05       0    4996     .05       0  5047.1     .12       0
  5355.8     .16       0  5575.3      .1       0  5689.1     .05       0
  5794.8      .1       0
Bank Sta=4945,5027
XS Rating Curve= 0 ,0
Exp/Cntr=0.3,0.1

Type RM Length L Ch R = 1 ,26431   ,619,619,619
BEGIN DESCRIPTION:
BAYOU CREEK 37.0
END DESCRIPTION:
XS GIS Cut Line= 3
      2368372.98      13210284.6      2367591.74     13209930.43
      2366268.84     13209430.44
#Sta/Elev= 30
  4324.8  110.36  4440.4  106.18  4449.2  105.35  4500.9  102.84  4923.5   76.72
  4961.5   75.83  4967.4   76.43  4978.4   75.07  5000.1   63.54  5003.3   64.04
  5013.2   64.75  5030.8   75.67  5044.2   75.85  5174.8   76.44  5210.2   69.66
  5283.1   75.83  5295.4   69.74  5314.9   75.44  5350.4   76.62  5460.4    77.3
  5465.8   70.98  5496.9   76.39  5614.5    77.8  5655.6   72.06  5691.2   77.81
  6117.1   86.85    6142   87.69    6288   93.12  6587.3   98.92  6596.8    98.8
#Mann= 15 ,-1 , 0
  4324.8     .05       0  4440.4      .1       0  4449.2     .16       0
  4500.9      .1       0  4923.5     .05       0  4961.5      .1       0
  5003.3     .07       0  5013.2      .1       0  5030.8     .12       0
  5350.4      .1       0  5614.5     .12       0  6117.1      .1       0
    6142     .12       0    6288      .1       0  6587.3     .05       0
Bank Sta=4967.4,5044.2
XS Rating Curve= 0 ,0
Exp/Cntr=0.3,0.1

Type RM Length L Ch R = 1 ,25812   ,415,415,415
BEGIN DESCRIPTION:
BAYOU CREEK 36.0
END DESCRIPTION:
XS GIS Cut Line= 3
      2368575.26       13209459.      2368186.32     13209507.62
      2366861.33     13209160.76
#Sta/Elev= 30
  4378.6   99.26  4416.4  100.52  4577.7  101.08  4688.5   98.17    4749   94.78
  4800.1   89.61  4820.8   89.31  4841.5   84.96    4875   82.21  4903.5   78.01
  4910.2   75.76  4934.5   74.02  4975.9   75.23  4985.9   70.39  4991.1    67.4
  5006.6   66.52  5009.9   67.02  5026.3   75.18  5037.9   76.33  5089.6   73.13
    5286   77.36  5575.4   76.47  5637.4   76.01  5657.5   77.57  5751.1   77.58
  5778.7   78.35  5854.4   79.27  6050.9      85  6061.7    86.5  6140.2   89.61
#Mann= 10 ,-1 , 0
  4378.6     .05       0  4416.4      .1       0  4985.9     .07       0
  4991.1      .1       0  5009.9     .12       0    5286      .1       0
  5575.4     .12       0  5751.1      .1       0  5778.7     .05       0
  5854.4      .1       0
Bank Sta=4910.2,5037.9
XS Rating Curve= 0 ,0
Exp/Cntr=0.3,0.1

Type RM Length L Ch R = 1 ,25397   ,492,492,492
BEGIN DESCRIPTION:
BAYOU CREEK 35.0
END DESCRIPTION:
XS GIS Cut Line= 3
      2368658.55     13209375.67      2368394.66     13209090.95
      2366931.03     13209007.71
#Sta/Elev= 30
    4335   92.38  4398.6   90.49  4462.1   89.11  4504.6   85.85  4561.3   82.41
  4632.2   78.54  4740.2   76.62  4830.3   76.35  4870.4   75.66  4940.5    73.9
  4970.5   75.68  4980.6   69.52  5000.3   65.17  5003.6   65.67  5010.6   68.54
  5020.6   75.13  5030.6   76.12  5090.7   75.88  5130.8   73.22  5200.9   72.95
  5341.1   76.23  5371.2   75.29    5414   76.39  5511.4   76.12  5611.6   74.63
  5641.6   76.01  5811.9   78.91    5862   81.58  5912.1   82.18  6189.2   89.64
#Mann= 15 ,-1 , 0
    4335     .05       0  4398.6      .1       0  4504.6     .16       0
  4561.3      .1       0  4740.2     .16       0  4870.4      .1       0
  5003.6     .07       0  5010.6      .1       0  5130.8     .12       0
  5371.2      .1       0    5414     .12       0  5511.4      .1       0
  5641.6     .12       0  5811.9     .05       0  5912.1      .1       0
Bank Sta=4830.3,5030.6
XS Rating Curve= 0 ,0
Exp/Cntr=0.3,0.1

Type RM Length L Ch R = 1 ,24905   ,1008,1008,1008
BEGIN DESCRIPTION:
BAYOU CREEK 34.0
END DESCRIPTION:
XS GIS Cut Line= 3
      2368818.24     13208590.95      2368082.16     13208618.73
      2366915.46     13208945.12
#Sta/Elev= 30
  4433.6  100.93  4444.1   98.66  4453.4   98.51  4464.1  101.39  4514.2  101.47
  4664.3   94.62  4721.1   88.21  4814.4   80.47  4874.4   75.96  4964.5   72.85
  4974.5   66.79  4983.5   63.61  4986.8   64.11  4988.8   65.87    4992   65.08
  5004.5   65.16  5014.5   75.45  5064.6   76.39  5114.6   74.14  5254.4   73.56
  5309.8   72.12  5361.7   73.68  5610.9    75.6  5734.5   73.86  5797.9    74.2
  5870.5   75.98  5974.4   80.54  6026.3   82.66  6213.2   85.82  6381.7   90.45
#Mann= 9 ,-1 , 0
  4433.6     .05       0  4514.2     .16       0  4814.4      .1       0
    4992     .07       0  5004.5      .1       0  5014.5     .12       0
  5254.4      .1       0  5361.7     .05       0  5974.4      .1       0
Bank Sta=4874.4,5014.5
XS Rating Curve= 0 ,0
Exp/Cntr=0.3,0.1

Type RM Length L Ch R = 1 ,23897   ,584,584,584
BEGIN DESCRIPTION:
BAYOU CREEK 33.0
END DESCRIPTION:
XS GIS Cut Line= 3
      2368693.26     13207361.79      2368193.27     13207688.17
      2366812.32     13208791.54
#Sta/Elev= 30
    4533  101.63  4539.6  101.89  4554.5   95.83  4563.5   96.56  4569.6  101.88
  4575.6  102.82  4663.1   98.56  4792.8   93.55  4801.9   89.99    4823   88.55
  4859.2   92.01  4916.5    92.7  4945.6   92.67  4952.7   87.26  4973.8   78.28
  4981.5   70.55  4994.9   68.17  5004.1   64.52  5009.8   63.91  5017.3   65.56
  5025.2   73.68  5040.3   73.63  5168.6   72.71  5381.5   74.21  5552.8   72.07
  5581.7   72.47    6158   73.42  6286.1   78.22  6442.8   85.49  6897.7   95.35
#Mann= 10 ,-1 , 0
    4533     .05       0  4663.1      .1       0  4916.5     .12       0
  4994.9     .07       0  5004.1     .12       0  5168.6     .16       0
  5381.5     .05       0  5552.8     .16       0  5581.7     .05       0
  6286.1      .1       0
Bank Sta=4973.8,5040.3
XS Rating Curve= 0 ,0
Exp/Cntr=0.3,0.1

Type RM Length L Ch R = 1 ,23313   ,449,449,449
BEGIN DESCRIPTION:
BAYOU CREEK 32.0
END DESCRIPTION:
XS GIS Cut Line= 3
       2368412.1     13207069.23      2367512.32     13207694.96
      2366644.27     13208675.85
#Sta/Elev= 30
  4328.1  104.27    4488  101.59  4565.7  100.17  4601.5   99.22  4738.5   92.48
  4783.1   89.64  4845.9   80.52  4905.3   74.63  4918.1   73.62  4968.1   71.72
  4976.8   71.61  4991.2   65.27  4997.5   63.95  5000.8   64.45  5012.6   65.45
  5018.7   69.71  5048.4   73.26  5054.5   72.78  5105.1   71.11  5134.8    73.2
  5198.2   71.67  5227.3   71.32    5320   69.47  5423.8   72.35  5527.9   72.94
  5711.9   71.14  5960.4   75.94  6087.5   79.23  6519.9   94.62  6733.9   97.38
#Mann= 13 ,-1 , 0
  4328.1     .05       0    4488     .05       0  4565.7      .1       0
  4601.5     .05       0  4738.5      .1       0  4845.9     .05       0
  4905.3      .1       0  4968.1     .05       0  5000.8     .04       0
  5012.6     .05       0  5198.2     .12       0  5227.3     .05       0
  5960.4      .1       0
Bank Sta=4918.1,5054.5
XS Rating Curve= 0 ,0
Exp/Cntr=0.3,0.1

Type RM Length L Ch R = 1 ,22864   ,597,597,597
BEGIN DESCRIPTION:
BAYOU CREEK 31.0
END DESCRIPTION:
XS GIS Cut Line= 4
       2368179.4     13206945.11       2367714.1     13207111.78
      2366755.77     13207840.95      2366658.55     13208410.36
#Sta/Elev= 30
  4155.6  100.11    4338   95.37  4589.2   86.38  4729.8   78.76    4786   77.27
  4829.6   72.58  4858.7    72.6  4879.5   72.97  4921.7   70.38    4972   71.57
  4979.3   71.19  4985.6   63.53  5000.1   63.47  5008.1   62.86  5011.4   63.36
  5014.6   70.91  5035.5      71  5108.2   68.08  5158.1    69.1    5208   71.87
  5278.7   71.72  5343.1    69.5  5600.3   73.42  5686.2   75.45  5880.3   83.66
  5981.8   85.37    6134   90.03  6357.1   93.67  6397.7    94.9  6431.7   95.47
#Mann= 12 ,-1 , 0
  4155.6     .05       0    4338     .05       0  4589.2      .1       0
  4858.7     .12       0  5000.1     .07       0  5008.1     .12       0
  5158.1      .1       0  5278.7     .12       0  5600.3     .16       0
    6134      .1       0  6357.1     .16       0  6397.7      .1       0
Bank Sta=4972,5035.5
XS Rating Curve= 0 ,0
Exp/Cntr=0.3,0.1

Type RM Length L Ch R = 1 ,22267   ,377,377,377
BEGIN DESCRIPTION:
BAYOU CREEK 30.0
END DESCRIPTION:
XS GIS Cut Line= 3
      2368227.99     13206757.61      2367346.04     13206924.28
      2366214.06     13207340.96
#Sta/Elev= 30
  3665.5  100.97  3818.4   97.29  4066.5   90.58  4429.1   75.91  4611.6   72.54
  4697.6   68.75  4758.5   71.21  4900.2   69.98    4936   68.43  4976.9   70.32
  4991.6    68.9  4998.2   61.97  5005.8   60.95  5008.6   60.45  5011.8   60.95
  5016.7    66.9    5022   69.65  5047.1    70.3    5158   67.63  5243.3   71.87
  5341.1   77.59  5427.1   80.84    5467   84.49  5477.4   83.61  5513.2   86.73
  5552.3   88.65  5629.7   93.01  5679.9   93.83  5701.5   95.49  5769.3   97.86
#Mann= 9 ,-1 , 0
  3665.5     .05       0  3818.4     .05       0  4066.5      .1       0
  4611.6     .12       0  5005.8     .12       0  5243.3     .16       0
    5467      .1       0  5552.3     .16       0  5701.5      .1       0
Bank Sta=4976.9,5047.1
XS Rating Curve= 0 ,0
Exp/Cntr=0.3,0.1

Type RM Length L Ch R = 1 ,21890   ,647,647,647
BEGIN DESCRIPTION:
BAYOU CREEK 29.0
END DESCRIPTION:
XS GIS Cut Line= 4
      2368464.07     13206577.06      2367748.82     13206570.12
      2366200.21     13206965.95      2365931.06     13207076.37
#Sta/Elev= 30
  3137.2  101.84  3223.6  102.27  3363.6  100.26  3413.6   99.45  3473.6   96.34
  3563.6   97.96  3803.6   92.09  3925.9   87.31  4111.7   77.47  4256.2   72.82
  4648.4   69.78  4772.2   70.86  4869.7    69.2  4875.4   70.16  4910.5   69.33
  4927.1   70.87    4958   70.24  4968.3    68.5  4991.9   59.98  4995.2   60.48
  4999.3   60.78    5020   68.01  5068.7   68.27  5081.9   71.05  5155.5   78.31
    5278   87.52  5339.9   91.84  5395.3   93.67  5521.5  100.42  5741.8  105.18
#Mann= 8 ,-1 , 0
  3137.2     .05       0  3363.6     .05       0  3803.6      .1       0
  4648.4     .12       0  4995.2     .07       0  4999.3     .12       0
    5278      .1       0  5521.5     .05       0
Bank Sta=4958,5081.9
XS Rating Curve= 0 ,0
Exp/Cntr=0.3,0.1

Type RM Length L Ch R = 1 ,21243   ,129,129,129
BEGIN DESCRIPTION:
BAYOU CREEK 28.0
END DESCRIPTION:
XS GIS Cut Line= 4
      2368296.15      13206470.9      2367674.51     13206333.34
      2366268.26     13206286.47      2365674.55     13206036.48
#Sta/Elev= 30
  3081.7  101.47  3192.8   99.78  3445.6   96.77  3551.2   94.36  3653.6   90.95
  3745.2   87.22  3895.3   78.71  4095.4   72.16  4455.6   68.39  4635.7   71.12
  4705.7   67.47  4945.8   70.06  4967.3   68.43  4992.9    61.9  4995.6    61.4
  5035.9   67.47  5045.9    72.1  5115.9   80.02  5123.2   85.52  5340.5   88.12
  5345.9   91.11  5393.4   91.33  5398.8   94.46  5446.3   94.01  5451.7   97.78
  5493.8   97.68  5499.2  101.49  5546.7  100.37  5552.1  103.76  5769.6  102.02
#Mann= 8 ,-1 , 0
  3081.7     .05       0  3192.8     .05       0  3445.6     .08       0
  3551.2     .05       0  3653.6     .08       0  3745.2     .05       0
  4992.9     .04       0  4995.6     .05       0
Bank Sta=4945.8,5045.9
XS Rating Curve= 0 ,0
Exp/Cntr=0.3,0.1

Type RM Length L Ch R = 1 ,21114   ,521,521,521
BEGIN DESCRIPTION:
Mapping XS 8d302372
END DESCRIPTION:
XS GIS Cut Line= 4
      2368438.89     13206390.85      2367653.68     13206203.13
      2366299.51     13206161.47      2365742.45     13205948.01
#Sta/Elev= 30
  2936.5   101.1  3040.5   98.44  3237.1   95.44  3544.3   92.43  3698.5   88.83
  3809.8    82.9  4039.9   70.78  4620.2   68.25  4730.3      68  4850.3   70.79
  4930.4   68.05  4960.4   69.88  4980.4   69.76  5000.1   60.15  5003.4   60.65
  5010.4   61.73  5020.4   63.15  5030.4   66.19  5040.4    64.9  5060.4   69.97
  5080.4   72.67  5085.7   77.46  5090.7   76.01  5111.3   81.22  5151.1   85.86
  5156.5   84.58  5181.1   89.02  5211.2   89.29  5430.1     107  5695.2   106.3
#Mann= 12 ,-1 , 0
  2936.5     .05       0  3040.5     .08       0  3237.1     .05       0
  3544.3     .08       0  3809.8     .05       0  4620.2      .1       0
  4730.3     .12       0  5003.4     .07       0  5010.4     .12       0
  5020.4      .1       0  5111.3     .12       0  5211.2     .05       0
Bank Sta=4960.4,5060.4
XS Rating Curve= 0 ,0
Exp/Cntr=0.3,0.1

Type RM Length L Ch R = 1 ,20593   ,441,441,441
BEGIN DESCRIPTION:
BAYOU CREEK 27.0
END DESCRIPTION:
XS GIS Cut Line= 3
      2368454.52     13206312.73      2366486.41     13205721.85
      2366086.41     13205721.85
#Sta/Elev= 30
  2998.1   99.48  3318.9   91.28  3489.4    90.1  3593.7   91.04  3764.2    87.6
    4018   73.81  4153.9      69  4286.1   68.03  4487.8   69.28  4717.5   66.01
  4790.6    66.3  4853.2   68.73  4945.3   67.04  4978.4   68.85  4983.6   62.65
  4999.4   59.04  5016.4   58.02  5019.7   58.52  5021.9    63.7  5030.7   68.11
  5049.5   69.01  5101.7   70.46  5131.7   74.47  5181.7   77.01  5191.7   78.26
  5201.7   81.97  5211.7   88.11  5281.7   96.07  5361.7  102.17    5453   105.8
#Mann= 9 ,-1 , 0
  2955.9     .05       0  3915.8      .1       0  4037.3     .05       0
  4597.6      .1       0  4754.9     .12       0  4997.3     .07       0
  5003.3     .12       0  5070.2      .1       0  5323.2     .05       0
Bank Sta=4978.4,5049.5
XS Rating Curve= 0 ,0
Exp/Cntr=0.3,0.1

Type RM Length L Ch R = 1 ,20152   ,529,529,529
BEGIN DESCRIPTION:
Mapping XS 473ce4c6
END DESCRIPTION:
XS GIS Cut Line= 4
      2368626.41     13206271.07      2367190.14     13205578.13
       2366669.3     13205421.88      2366152.56     13205661.62
#Sta/Elev= 30
  3101.2  103.22  3283.2   96.42  3582.7   88.69  3746.5   81.85  3814.4   82.81
    3837   86.89  3843.6   89.62    3854   89.81  3859.6   89.54  3865.9   86.62
  3888.1   81.98  3910.3   80.66  4023.4   79.15  4272.1   72.15    4645   67.45
  4754.2    69.1  4792.5   66.38  4834.1   65.35  4957.8   66.01  4996.1   61.81
  4998.3   58.47    5001   57.97  5022.1   62.55  5034.3   67.85  5053.4   66.27
  5074.3    69.5  5095.1   71.51  5171.8   74.03  5615.2    98.1  5809.3   105.5
#Mann= 12 ,-1 , 0
  3015.6     .05       0  3730.9      .1       0  4070.6     .12       0
    4081      .1       0    4187     .05       0  4307.3      .1       0
  4401.9     .05       0  4819.6     .12       0  4998.6     .07       0
  5004.6     .12       0  5129.8      .1       0  5645.7     .05       0
Bank Sta=4754.2,5074.3
XS Rating Curve= 0 ,0
Exp/Cntr=0.3,0.1

Type RM Length L Ch R = 1 ,19623   ,520,520,520
BEGIN DESCRIPTION:
Mapping XS 7470d99e
END DESCRIPTION:
XS GIS Cut Line= 4
      2368466.16      13204927.1      2367804.72     13205338.55
      2367070.35     13205192.72      2366152.54     13205630.38
#Sta/Elev= 30
  3707.4  108.45  3764.4  107.11  3858.7  102.91  3908.7  102.99  3966.5  100.15
  4076.3   97.79    4244   90.23    4323   89.92    4460   84.87  4666.8   69.33
  4724.5   66.63  4819.8   66.25  4962.5   67.97  4985.4   64.09  4993.1   59.34
  5000.3   58.99    5003   58.49  5031.5   66.87  5115.4   65.95  5329.1   67.71
  5448.5   69.35  5584.3   73.73  5646.8   77.68  5697.7   78.52  5765.8   81.81
  5788.5   84.28  5891.6   90.21    6080   99.21  6201.8  103.51  6251.9  105.29
#Mann= 9 ,-1 , 0
  3707.4     .05       0  3764.4     .05       0  3966.5      .1       0
  4666.8     .16       0  4819.8     .12       0  4993.1     .07       0
  5000.3     .12       0  5329.1      .1       0  6201.8     .05       0
Bank Sta=4962.5,5031.5
XS Rating Curve= 0 ,0
Exp/Cntr=0.3,0.1

Type RM Length L Ch R = 1 ,19103   ,496,496,496
BEGIN DESCRIPTION:
Mapping XS 5216ed63
END DESCRIPTION:
XS GIS Cut Line= 3
      2368480.57     13204870.02      2367365.97     13204745.02
      2366139.38     13205619.17
#Sta/Elev= 30
  3999.4  110.54  4062.6  109.53  4263.9  106.84  4384.7  102.09  4520.9   93.54
  4535.6    94.3  4646.3   82.45  4777.1   66.72  4817.4   64.49  4837.5   61.48
  4876.4   64.45  4938.1   65.97  4966.6   64.78  4978.4   58.07  4988.4    56.6
  4995.5   56.55  4998.2   56.05  5001.5   56.55  5008.5   63.76  5018.6   66.25
  5068.9   63.77  5149.8   66.95  5342.8   66.13  5773.1   69.63  5873.9   73.16
  6016.5   81.19  6174.9   85.65  6268.5   91.88  6526.7  102.59  6627.2  105.84
#Mann= 10 ,-1 , 0
  3999.4     .05       0  4062.6     .05       0  4263.9      .1       0
  4646.3     .12       0  4777.1      .1       0  4837.5     .12       0
  4988.4     .07       0  4995.5     .12       0  5342.8      .1       0
  6526.7     .05       0
Bank Sta=4938.1,5018.6
XS Rating Curve= 0 ,0
Exp/Cntr=0.3,0.1

Type RM Length L Ch R = 1 ,18607   ,103,103,103
BEGIN DESCRIPTION:
BAYOU CREEK 26.0
END DESCRIPTION:
XS GIS Cut Line= 4
      2368470.16     13204797.12       2367824.3      13204172.1
      2367355.55     13204390.85      2366128.97     13205580.97
#Sta/Elev= 30
    3777  112.02  3948.5  109.81  4075.9  102.54  4203.2   97.54  4330.5      90
  4394.1   84.63  4662.9   74.84  4826.5   75.51  4841.9    74.8  4870.6   66.12
  4903.7   65.52  4961.7   65.49  4984.5   59.46    4989   55.76  4991.8   55.26
  5001.9   55.83  5014.1   62.94  5069.3   64.85  5098.8   61.75  5209.9   66.45
  5471.5   63.73  5478.7   59.81  5499.8    58.2  5535.3   64.32    5606   65.81
  6001.9   68.58    6405   84.82  6772.8  101.08  6836.4  103.34  6902.1  105.66
#Mann= 12 ,-1 , 0
    3777     .05       0  3948.5     .05       0  4075.9      .1       0
  4203.2     .05       0  4330.5      .1       0  4903.7     .12       0
  4984.5     .07       0    4989     .12       0  5471.5      .1       0
    6405     .05       0  6772.8      .1       0  6836.4     .05       0
Bank Sta=4961.7,5069.3
XS Rating Curve= 0 ,0
Exp/Cntr=0.3,0.1

Type RM Length L Ch R = 1 ,18504   ,537,537,537
BEGIN DESCRIPTION:
BAYOU CREEK 25.0
END DESCRIPTION:
XS GIS Cut Line= 2
      2368706.16     13203242.54      2365893.78     13205482.02
#Sta/Elev= 30
  3403.9  111.29  3568.9   112.8    4011   108.4  4159.9  103.27  4267.2   97.41
  4416.2    81.6  4494.6   77.87  4537.9   79.09  4593.9   73.49  4701.3   69.57
  4829.4   67.28  4843.8    67.2  4928.7   65.98  4957.5    64.5  4999.5   56.07
  5007.2      57  5021.6   58.63    5028   62.66  5042.4   64.89  5106.5   62.43
  5213.8   66.17  5327.5   65.81    5462    63.1  5484.4   63.36  5732.7   65.98
  6003.4   69.84  6280.4    81.1  6515.9   92.28  6751.1   99.63    6999  104.54
#Mann= 15 ,-1 , 0
  3403.9     .05       0  3568.9      .1       0  4701.3     .12       0
  4829.4     .05       0  4843.8     .12       0  5007.2     .07       0
  5021.6     .12       0  5213.8      .1       0  5327.5     .12       0
    5462      .1       0  5484.4     .12       0  5732.7      .1       0
  6280.4     .05       0  6515.9      .1       0  6751.1     .05       0
Bank Sta=4928.7,5042.4
XS Rating Curve= 0 ,0
Exp/Cntr=0.3,0.1

Type RM Length L Ch R = 1 ,17967   ,313,313,313
BEGIN DESCRIPTION:
Mapping XS e15a9df4
END DESCRIPTION:
XS GIS Cut Line= 2
       2368718.7     13202640.57      2365288.14     13205307.25
#Sta/Elev= 30
    2847  105.36  2994.8  101.15  3030.1   98.07  3073.5   96.49  3094.4   93.37
  3108.8    94.4  3115.2   91.56  3129.7   90.58  3173.1   91.84  3450.9   84.18
  4249.1   71.92  4669.9   69.19  4912.4   67.53  4962.2      66  4989.4   58.07
    5012   57.52  5018.1   56.73  5026.5   57.58  5032.8   60.64  5076.2   61.09
  5090.1   65.58    5132    66.8  5310.6   68.18  5567.6   69.85  6222.8   76.67
  6707.9   91.44  6892.5   88.07  7099.7   90.99  7155.8   90.44  7192.1   91.19
#Mann= 11 ,-1 , 0
    2847     .05       0  3030.1     .08       0  4249.1     .05       0
  4669.9     .08       0    5012     .08       0  5026.5     .05       0
  5076.2     .08       0  5310.6     .05       0  5567.6     .08       0
  7099.7      .1       0  7155.8     .08       0
Bank Sta=4912.4,5132
XS Rating Curve= 0 ,0
Exp/Cntr=0.3,0.1

Type RM Length L Ch R = 1 ,17654   ,649,649,649
BEGIN DESCRIPTION:
BAYOU CREEK 24.0
END DESCRIPTION:
XS GIS Cut Line= 2
      2368568.98     13202478.23      2365118.47     13205158.35
#Sta/Elev= 30
  2652.6  112.35  2837.8  109.51  2995.3  106.82  3179.9   97.02  3287.3   91.77
  3607.1   87.74  3750.1   93.57    4142   72.57  4235.2    76.8  4305.8   90.58
  4384.5    84.2  4761.9   69.35  4890.5   66.88  4896.8   67.18  4969.2   59.91
  4996.4    52.3  5004.5   53.59  5010.8   58.33  5025.3   61.94  5139.4   63.17
  5153.8   64.35  5325.8   59.49  5574.7   70.66  5638.9   72.87  5788.3   75.11
    5959   79.51  6115.9   81.61  6308.7   81.55  6921.3   97.61  7021.7   98.79
#Mann= 19 ,-1 , 0
  2652.6     .05       0  2837.8     .05       0  2995.3      .1       0
  3179.9      .1       0  3287.3      .1       0  4384.5     .05       0
  4761.9      .1       0  4890.5     .12       0  5004.5     .07       0
  5010.8     .12       0  5025.3     .12       0  5139.4      .1       0
  5574.7     .16       0  5638.9      .1       0  5788.3      .1       0
    5959      .1       0  6115.9      .1       0  6308.7     .05       0
  6921.3     .05       0
#XS Ineff= 2 , 0
         4328.41    89.4
Permanent Ineff=
       F       F
Bank Sta=4896.8,5153.8
XS Rating Curve= 0 ,0
Exp/Cntr=0.3,0.1
