--- UNT 020 IN LACR.prj (project) ---

Proj Title=UNT 020 IN LACR Base Level Engineering
Current Plan=p01
Default Exp/Contr=0.3,0.1
English Units
Geom File=g01
Flow File=f01
Plan File=p01
Y Axis Title=Elevation
X Axis Title(PF)=Main Channel Distance
X Axis Title(XS)=Station
BEGIN DESCRIPTION:
UNT 020 IN LACR
END DESCRIPTION:
DSS Export Rating Curves= 0
DSS Export Rating Curve Sorted= 0
DSS Export Volume Flow Curves= 0
DXF OffsetX= 0
DXF OffsetY= 0
DXF ScaleX= 1
DXF ScaleY= 10

--- UNT 020 IN LACR.p01 (plan) ---

Plan Title=Multiple Run
Short Identifier=Multiple
Geom File=g01
Flow File=f01
Subcritical Flow
K Sum by GR= 0
Std Step Tol= 0.01
Critical Tol= 0.01
Num of Std Step Trials= 20
Max Error Tol= 0.3
Flow Tol Ratio= 0.001
Split Flow NTrial= 30
Split Flow Tol= 0.02
Split Flow Ratio= 0.02
Log Output Level= 0
Friction Slope Method= 1
Unsteady Friction Slope Method= 2
Unsteady Bridges Friction Slope Method= 1
Parabolic Critical Depth
Global Vel Dist=  1 , 1 , 1
Global Log Level= 0
CheckData=True
Encroach Param= -1, 0, 0, 0
BEGIN DESCRIPTION:
Multiple Run
END DESCRIPTION:

--- UNT 020 IN LACR.f01 (steady flow) ---

Flow Title=Multiple
Program Version=4.10
Number of Profiles= 7
Profile Names=10-year,25-year,50-year,1pct_min,100-year,1pct_plu,500-year
River Rch & RM=UNT 020 IN LACR,Reach-1         ,41268
     337     485     612     568     768    1038    1229
River Rch & RM=UNT 020 IN LACR,Reach-1         ,35580
     429     624     793     741    1003    1356    1628
River Rch & RM=UNT 020 IN LACR,Reach-1         ,35306
     468     682     868     811    1097    1484    1784
River Rch & RM=UNT 020 IN LACR,Reach-1         ,33266
     468     682     868     811    1097    1484    1784
River Rch & RM=UNT 020 IN LACR,Reach-1         ,32634
     468     682     868     811    1097    1484    1784
River Rch & RM=UNT 020 IN LACR,Reach-1         ,31299
     608     896    1149    1082    1463    1978    2411
River Rch & RM=UNT 020 IN LACR,Reach-1         ,30675
     608     896    1149    1082    1463    1978    2411
River Rch & RM=UNT 020 IN LACR,Reach-1         ,29742
     700    1038    1337    1263    1708    2309    2835
River Rch & RM=UNT 020 IN LACR,Reach-1         ,28409
     810    1205    1556    1473    1992    2693    3320
River Rch & RM=UNT 020 IN LACR,Reach-1         ,27471
     810    1205    1556    1473    1992    2693    3320
River Rch & RM=UNT 020 IN LACR,Reach-1         ,26989
     810    1205    1556    1473    1992    2693    3320
River Rch & RM=UNT 020 IN LACR,Reach-1         ,22844
     860    1279    1650    1559    2109    2852    3506
River Rch & RM=UNT 020 IN LACR,Reach-1         ,16899
     881    1310    1690    1597    2160    2921    3590
River Rch & RM=UNT 020 IN LACR,Reach-1         ,15537
     881    1310    1690    1597    2160    2921    3590
River Rch & RM=UNT 020 IN LACR,Reach-1         ,14329
    1004    1496    1932    1828    2472    3343    4115
River Rch & RM=UNT 020 IN LACR,Reach-1         ,8472
    1049    1564    2021    1912    2586    3497    4308
River Rch & RM=UNT 020 IN LACR,Reach-1         ,4001
    1047    1558    2011    1901    2571    3477    4274
Boundary for River Rch & Prof#=UNT 020 IN LACR,Reach-1         , 1
Up Type= 0
Dn Type= 3
Dn Slope=0.0017
Boundary for River Rch & Prof#=UNT 020 IN LACR,Reach-1         , 2
Up Type= 0
Dn Type= 3
Dn Slope=0.0017
Boundary for River Rch & Prof#=UNT 020 IN LACR,Reach-1         , 3
Up Type= 0
Dn Type= 3
Dn Slope=0.0017
Boundary for River Rch & Prof#=UNT 020 IN LACR,Reach-1         , 4
Up Type= 0
Dn Type= 3
Dn Slope=0.0017
Boundary for River Rch & Prof#=UNT 020 IN LACR,Reach-1         , 5
Up Type= 0
Dn Type= 3
Dn Slope=0.0017
Boundary for River Rch & Prof#=UNT 020 IN LACR,Reach-1         , 6
Up Type= 0
Dn Type= 3
Dn Slope=0.0017
Boundary for River Rch & Prof#=UNT 020 IN LACR,Reach-1         , 7
Up Type= 0
Dn Type= 3
Dn Slope=0.0017
DSS Import GetInterval= 0
DSS Import GetPeak= 0
DSS Import FillOption= 0

--- UNT 020 IN LACR.g01 (geometry) ---

Geom Title=Existing Conditions
Program Version=4.10

River Reach=UNT 020 IN LACR ,Reach-1
Reach XY= 30
      2166587.72     13192796.86      2167237.72     13193146.86
      2168137.72     13192646.86      2170637.72     13192896.85
      2173837.72     13193896.85      2175587.72     13194996.85
      2176787.72     13194946.86      2178487.72     13195796.85
      2179187.72     13196446.85      2179187.72     13197246.86
      2179737.72     13197646.85      2179837.72     13199046.86
      2180387.72     13200496.85      2181337.72     13201146.85
      2181587.72     13202146.86      2182537.72     13202596.85
      2182387.72     13203296.86      2182737.72     13204196.85
      2182387.72     13205446.86      2183137.72     13205896.85
      2183037.72     13206596.86      2183387.72     13207146.85
      2184187.72     13208046.86      2184937.72     13207596.85
      2186237.72     13208696.85      2187537.72     13208496.85
      2187787.72     13209646.85      2188687.72     13209146.85
      2189487.72     13210396.85      2191387.72     13211046.85

Type RM Length L Ch R = 1 ,41268   ,586,586,586
BEGIN DESCRIPTION:
UNT 020 IN LACR 75.0
END DESCRIPTION:
XS GIS Cut Line= 3
      2166573.55     13193687.29        2166893.     13192333.09
      2166816.62     13192013.66
#Sta/Elev= 30
  4136.5   522.1  4259.3   518.5  4354.3  514.99  4383.5   514.8  4507.5  511.22
  4578.7  509.88  4671.2  508.93  4677.9  508.62  4712.3  508.56  4732.9  509.32
  4745.5  508.62    4774  508.68  4842.9  507.47  4845.6  506.97  4848.9  507.47
  4926.5  507.61  4992.9  507.87  5030.8  507.83  5094.4  509.15  5102.7  509.18
    5113  508.38  5128.2  508.83  5173.9  509.77  5205.5  511.14  5221.3  512.37
  5252.6  513.09  5395.8  517.66  5527.3   519.7  5678.2  523.39  5856.3  526.54
#Mann= 9 ,-1 , 0
  4136.5     .05       0  4507.5      .1       0  4677.9     .12       0
  4842.9     .07       0  4848.9     .12       0  4926.5     .16       0
  4992.9     .12       0  5128.2     .16       0  5252.6     .05       0
Bank Sta=4671.2,5128.2
XS Rating Curve= 0 ,0
Exp/Cntr=0.3,0.1

Type RM Length L Ch R = 1 ,40682   ,382,382,382
BEGIN DESCRIPTION:
UNT 020 IN LACR 74.0
END DESCRIPTION:
XS GIS Cut Line= 4
      2167018.01     13193819.19      2167233.28     13193395.59
      2167240.22     13192583.09      2167095.11     13192320.51
#Sta/Elev= 30
  4273.8  519.97  4283.1  520.17  4305.4  519.07  4431.3  517.07  4527.9  516.06
  4700.3  512.68  4937.7  506.36  4977.7  505.64  5014.7   504.1  5017.5   503.6
  5020.7   504.1  5032.4  504.36  5117.7  505.42  5147.7  504.75  5227.7  506.29
  5288.5  507.72  5417.7  508.98  5437.7   509.7  5457.7  509.22  5487.7  509.31
  5507.7   510.2  5537.7   509.4  5561.5  509.78  5603.1  511.15  5625.7  511.06
  5700.5  513.56  5738.3  514.03  5781.9  515.72  5858.6  517.53  5861.5  517.62
#Mann= 7 ,-1 , 0
  4273.8      .1       0  4431.3     .05       0  5014.7     .03       0
  5020.7     .05       0  5032.4     .12       0  5288.5      .1       0
  5858.6     .05       0
Bank Sta=4937.7,5227.7
XS Rating Curve= 0 ,0
Exp/Cntr=0.3,0.1

Type RM Length L Ch R = 1 ,40300   ,539,539,539
BEGIN DESCRIPTION:
UNT 020 IN LACR 73.0
END DESCRIPTION:
XS GIS Cut Line= 4
      2167122.19     13193985.83      2167622.17      13193256.7
      2167476.34     13192374.75      2167254.09     13192048.34
#Sta/Elev= 30
  3953.9  521.63  4007.5  519.68  4136.1  516.57  4195.2  515.88  4488.8   508.9
  4524.6  508.33  4533.5  508.75  4539.5  508.01  4611.3  507.02  4697.9  505.61
  4826.5   505.3  4868.2  505.93  4989.9  503.13    5071  503.74  5162.2  502.97
  5172.3  503.57    5223  503.01  5232.9   502.2  5266.1  503.31  5444.2  504.25
  5476.4  505.26  5496.7  504.82  5587.9  506.47  5608.1  506.28  5627.4  507.17
  5795.5   512.2  5901.5  516.02  5922.9  517.42  5959.2  518.14  6126.8   524.5
#Mann= 4 ,-1 , 0
  3953.9      .1       0  4611.3     .07       0  5627.4      .1       0
  5795.5     .05       0
Bank Sta=4611.3,5627.4
XS Rating Curve= 0 ,0
Exp/Cntr=0.3,0.1

Type RM Length L Ch R = 1 ,39761   ,242,242,242
BEGIN DESCRIPTION:
UNT 020 IN LACR 72.0
END DESCRIPTION:
XS GIS Cut Line= 4
      2167303.22     13194006.46      2167761.56     13193103.66
      2168039.34     13192867.55       2167748.2     13192160.49
#Sta/Elev= 30
  3546.5  517.64  3685.9  514.19  3730.5  513.32  3941.8  509.04  4143.9  505.75
  4365.7  505.16  4455.6     506  4606.7  503.87  4789.4   502.3  4799.7  501.87
  4837.9  501.62  4866.5  498.25    4873  496.18  4880.8  496.36  4901.6   492.3
  4915.9  492.61  4920.2  490.94  4940.7  488.83  5010.6  486.43  5064.9  488.26
    5119  493.62  5148.5  500.17  5162.2  500.84  5201.6  500.37  5605.6  509.97
  5622.8  508.73  5646.8   509.2  5652.2  510.43  5670.5  509.84  5688.2  511.46
#Mann= 11 ,-1 , 0
  3546.5     .05       0  3685.9      .1       0  3730.5     .05       0
  3941.8      .1       0  4365.7     .05       0  4606.7     .12       0
  4789.4      .1       0  4799.7     .12       0  4837.9     .07       0
  5162.2     .12       0  5201.6      .1       0
Bank Sta=4837.9,5162.2
XS Rating Curve= 0 ,0
Exp/Cntr=0.3,0.1

Type RM Length L Ch R = 1 ,39519   ,265,265,265
BEGIN DESCRIPTION:
UNT 020 IN LACR 71.0
END DESCRIPTION:
XS GIS Cut Line= 4
      2167419.14     13194120.65      2167879.62     13193061.99
      2168147.98     13192990.96      2168187.72     13191896.85
#Sta/Elev= 30
  3223.6  517.82  3402.2  512.97  3500.4  511.63  3507.1  510.76  3565.8  509.35
  4060.9  503.96  4220.1  505.79    4351  504.54  4378.1  505.79    4415  510.04
  4438.2  510.73  4535.7  508.99  4570.7  509.16  4575.9  508.46    4611  508.98
  4709.8  507.68  4749.8  506.09  4779.9  506.42  4790.6  507.64  4919.9   507.1
    4980   506.2    5010  506.79    5070  506.41  5090.1  504.59  5110.1  501.35
  5129.8  499.85  5180.1  501.67  5290.2   502.8  5430.3  506.39  5750.5   517.4
#Mann= 3 ,-1 , 0
  3223.6      .1       0  4709.8     .07       0  4790.6      .1       0
#XS Ineff= 2 , 0
       0 4443.75  510.83 5065.91       0   506.8
Permanent Ineff=
       T       T
Bank Sta=4919.9,5010
XS Rating Curve= 0 ,0
Exp/Cntr=0.3,0.1

Type RM Length L Ch R = 1 ,39254   ,565,565,565
BEGIN DESCRIPTION:
UNT 020 IN LACR 70.0
END DESCRIPTION:
XS GIS Cut Line= 3
      2167787.75     13193996.82      2168414.34     13193096.72
      2168386.57     13191951.37
#Sta/Elev= 30
  3503.3  512.28  3607.1  509.55  3632.9  509.67  3740.2  507.48  3883.3   503.9
  3892.1  503.18  3898.2  503.61  3905.3  502.96  3967.6  502.33  4122.6  500.96
  4157.4  500.21  4228.9  500.98  4336.3  500.45  4351.1  501.07  4729.9  497.57
 4785.51  498.01    4930  497.63    4970  497.25  4989.7  496.36    5010  497.46
    5040  497.71    5050  498.25  5111.5  497.95    5130  497.75  5180.1     499
  5200.1  498.53  5380.1  501.46    5672  511.71  5720.2  513.65  5745.7  513.84
#Mann= 8 ,-1 , 0
  3503.3     .05       0  3607.1      .1       0  3967.6     .12       0
  4122.6      .1       0 4785.51     .07       0    5050     .12       0
  5111.5      .1       0    5672     .05       0
Bank Sta=4785.51,5040
XS Rating Curve= 0 ,0
Exp/Cntr=0.3,0.1

Type RM Length L Ch R = 1 ,38689   ,684,684,684
BEGIN DESCRIPTION:
UNT 020 IN LACR 69.0
END DESCRIPTION:
XS GIS Cut Line= 4
      2167979.98     13194164.45      2168748.19     13193422.27
      2169034.65     13192406.65      2168644.05     13191612.42
#Sta/Elev= 30
  3311.9  515.56    3441  512.27  3619.4  507.16  3630.9  506.68  3757.3     503
  3767.4  502.61  3888.6  499.37  4036.8  498.28  4052.5  498.08  4121.9  497.85
    4136  496.59  4193.1  495.87    4500  495.95  4644.6  494.88  4694.4  493.72
  4811.7  493.81  4872.2   494.7  4877.4   494.1  5009.1  493.74  5057.8  494.56
  5123.4  493.97    5620  501.88  5769.4  503.28    6047  510.39  6097.5  512.65
  6119.4  512.26  6159.3  514.21  6181.7  513.91  6215.4  515.29  6320.4  517.08
#Mann= 12 ,-1 , 0
  3311.9     .05       0    3441      .1       0  3619.4     .05       0
  3630.9      .1       0  3757.3     .05       0  3767.4      .1       0
  4036.8     .12       0  4052.5     .05       0  4193.1      .1       0
  4872.2     .07       0  5057.8      .1       0  6119.4     .05       0
Bank Sta=4872.2,5057.8
XS Rating Curve= 0 ,0
Exp/Cntr=0.3,0.1

Type RM Length L Ch R = 1 ,38005   ,646,646,646
BEGIN DESCRIPTION:
UNT 020 IN LACR 68.0
END DESCRIPTION:
XS GIS Cut Line= 3
       2169031.9     13194506.68      2169379.11      13193756.7
      2169684.66     13191805.34
#Sta/Elev= 30
    3202  506.82  3234.9  505.32  3245.9  505.32  3251.5  506.98    3334  504.93
  3611.8  504.83  3657.7  504.23  3675.1  502.45  3697.7  504.29  3829.9  498.52
  3846.5  499.43  3907.1  495.35  3929.1  496.79  3995.2  492.14  4012.5  493.64
  4025.6  491.99  4120.4  488.92  4129.5  489.89  4210.5  487.41  4342.1  489.14
  4483.5  486.87  4534.4  489.56    4919  491.51    5000  491.04  5010.1  491.09
  5546.6   498.3  5840.1  507.56  5863.6  506.45  5931.3  510.48  6003.6   512.6
#Mann= 3 ,-1 , 0
    3202      .1       0    4919     .07       0  5010.1      .1       0
#XS Ineff= 2 , 0
       0  4907.1  492.13               0
Permanent Ineff=
       T       F
Bank Sta=4919,5000
XS Rating Curve= 0 ,0
Exp/Cntr=0.3,0.1

Type RM Length L Ch R = 1 ,37359   ,610,610,610
BEGIN DESCRIPTION:
UNT 020 IN LACR 67.0
END DESCRIPTION:
XS GIS Cut Line= 3
      2169434.68     13194340.01      2170038.84     13193305.31
      2170205.28     13192050.07
#Sta/Elev= 30
  3389.8  498.98  3416.6  499.77  3445.5  497.98  3547.2  495.51  3578.6  496.57
  3590.3   495.1  3680.3  492.14  3701.8  493.48  3723.3  491.32  3766.3  490.15
    3825  488.61  3856.4  489.38  3868.2  488.12  3985.3  485.47  4001.1  486.36
    4044  484.57  4075.5  484.68    4088  483.05  4294.5  486.47  4556.6  486.99
    4698  488.59  4798.2  487.96    4918  489.28  4949.6  487.05  4979.8  484.97
  5010.1  486.64  5020.2  487.04  5153.2  486.79  5403.5  490.34  5854.2  502.02
#Mann= 3 ,-1 , 0
  3389.8     .12       0  4949.6     .07       0  5010.1      .1       0
#XS Ineff= 2 , 0
         4915.91  489.32
Permanent Ineff=
       F       F
Bank Sta=4949.6,5020.2
XS Rating Curve= 0 ,0
Exp/Cntr=0.3,0.1

Type RM Length L Ch R = 1 ,36749   ,490,490,490
BEGIN DESCRIPTION:
UNT 020 IN LACR 66.0
END DESCRIPTION:
XS GIS Cut Line= 4
      2169754.11     13194284.48      2170524.95     13193395.59
      2170795.78     13192624.75      2170684.68     13192103.97
#Sta/Elev= 30
  3343.8  490.96  3472.7  489.08  3614.2  485.86  3635.1  486.02  3755.7  482.71
  3777.5  481.85  3784.2  482.42  3862.1  482.75  3890.6  483.78  4414.8  482.73
  4457.5  482.86  4471.8  483.55  4506.9   482.9  4550.8  483.71  4575.7   483.2
  4656.8  483.92  4762.8  482.66  4921.8  482.42  4990.5  480.53  4993.3  480.03
  4996.5  480.53  5024.5  482.28    5049  482.87  5133.8  483.58  5303.4   486.3
  5774.9  498.48  5795.4  498.56    5826  500.14  5846.5  499.93  5869.9  500.74
#Mann= 3 ,-1 , 0
  3343.8      .1       0  4990.5     .07       0  4996.5      .1       0
Bank Sta=3755.7,5049
XS Rating Curve= 0 ,0
Exp/Cntr=0.3,0.1

Type RM Length L Ch R = 1 ,36259   ,679,679,679
BEGIN DESCRIPTION:
UNT 020 IN LACR 65.0
END DESCRIPTION:
XS GIS Cut Line= 4
      2169809.65       13194472.      2170774.95     13193562.25
      2171372.17     13192805.31      2171822.03      13192140.9
#Sta/Elev= 30
  3190.7   493.3  3228.5  492.54  3235.4  493.45  3270.6  491.69  3433.6  488.42
  3454.7  488.76    3483  487.65  3624.6  485.37  3638.8  485.86  3667.1  484.66
  3864.9  481.42  3978.2   480.7  4013.4  481.53  4162.3  481.89  4452.2  480.41
  4579.7  480.05  4629.4  481.04  4658.3  480.21  4786.6  481.05  4914.8  480.39
  4970.9  478.97  5096.2  478.41  5098.9  477.91  5102.2  478.41  5233.7  479.61
  5299.6   480.6  5331.6  480.78  5519.8  482.75  5829.7   487.4  6283.7  499.74
#Mann= 5 ,-1 , 0
  3190.7      .1       0  5096.2     .07       0  5102.2      .1       0
  5233.7     .12       0  5331.6      .1       0
Bank Sta=4452.2,5299.6
XS Rating Curve= 0 ,0
Exp/Cntr=0.3,0.1

Type RM Length L Ch R = 1 ,35580   ,274,274,274
BEGIN DESCRIPTION:
UNT 020 IN LACR 64.0
END DESCRIPTION:
XS GIS Cut Line= 3
       2170427.7     13194541.44      2171524.95     13193471.98
      2172351.31     13192395.63
#Sta/Elev= 30
  3226.8  490.78  3307.9     489  3336.2  487.38  3343.2  488.38  3477.6  485.26
  3484.6   484.5  3505.9  485.19  3647.2  482.16  3859.4  479.96  4090.2  478.73
  4227.5  478.54  4288.3  478.32  4495.9  477.96  4524.2  477.16  4582.7  477.24
  4743.4  477.86  4819.5  477.16  4896.4  477.32  4982.7  475.73  4985.4  475.23
  4988.7  475.73  5029.2  476.92  5106.2  476.61  5228.6  478.01  5413.5  481.84
  5762.2  493.62  5829.7  495.79  5870.3  497.46  5905.6  497.85    6116  506.31
#Mann= 11 ,-1 , 0
  3226.8      .1       0  4090.2     .12       0  4227.5      .1       0
  4288.3     .05       0  4582.7      .1       0  4819.5     .05       0
  4896.4      .1       0  4982.7     .07       0  4988.7      .1       0
  5762.2     .05       0  5829.7      .1       0
#XS Ineff= 2 , 0
         4742.55  477.86
Permanent Ineff=
       F       F
Bank Sta=4495.9,5228.6
XS Rating Curve= 0 ,0
Exp/Cntr=0.3,0.1

Type RM Length L Ch R = 1 ,35306   ,574,574,574
BEGIN DESCRIPTION:
UNT 020 IN LACR 63.0
END DESCRIPTION:
XS GIS Cut Line= 3
       2170608.3     13194596.96      2172288.84     13192992.81
      2172482.95     13192632.31
#Sta/Elev= 30
  3189.5  491.22  3270.6   489.6    3451  486.42  3507.3  483.65  3528.7   483.4
  3549.8  484.74  3620.5  482.11  3712.7  480.71  4009.6  479.21  4165.3  477.07
  4462.2  477.42  4518.8  475.44  4589.6  476.79  4808.8  476.52  4929.3  475.12
  4936.2  474.16  4950.3  475.05  5088.9  473.94  5091.6  473.44  5094.9  473.94
  5148.5  475.46  5194.8  476.48  5241.5  477.04  5334.5  478.63  5380.2   479.9
  5474.2  482.74  5517.6   484.1  5774.6  492.59  5878.4  498.39  5922.2  499.08
#Mann= 10 ,-1 , 0
  3189.5      .1       0  3270.6     .05       0  5088.9     .04       0
  5094.9     .05       0  5194.8      .1       0  5241.5     .05       0
  5334.5      .1       0  5380.2     .05       0  5474.2      .1       0
  5517.6     .05       0
#XS Ineff= 2 , 0
         4588.64  476.83
Permanent Ineff=
       F       F
Bank Sta=4518.8,5148.5
XS Rating Curve= 0 ,0
Exp/Cntr=0.3,0.1

Type RM Length L Ch R = 1 ,34732   ,468,468,468
BEGIN DESCRIPTION:
UNT 020 IN LACR 61.0
END DESCRIPTION:
XS GIS Cut Line= 3
      2171740.21       13194972.        2172643.     13193034.48
      2172629.13      13192701.5
#Sta/Elev= 30
  3327.3  487.22  3758.6  478.73    4176  472.36  4270.7   470.7  4336.9  470.31
  4367.3  471.12  4502.4  471.14  4524.5  472.59  4586.6  471.23  4810.8  471.97
  4849.2   470.7  4888.5  471.27  4940.7  470.12  4969.1  468.26  4986.5  469.83
  5006.3  464.49  5009.1  463.99  5012.3  464.49  5014.9   464.9  5020.9  468.33
  5037.7  471.14  5040.2  471.04    5089  472.13  5285.7  480.61  5346.1  481.73
  5374.5  483.93  5405.9  484.71    5453  486.21  5797.3  498.37  5798.1  498.41
#Mann= 10 ,-1 , 0
  3327.3      .1       0    4176     .12       0  4367.3      .1       0
  4810.8     .12       0  5006.3     .07       0  5012.3     .12       0
  5040.2      .1       0  5405.9     .05       0    5453      .1       0
  5797.3     .05       0
#XS Ineff= 2 , 0
         4522.16  472.52
Permanent Ineff=
       F       F
Bank Sta=4270.7,5037.7
XS Rating Curve= 0 ,0
Exp/Cntr=0.3,0.1

Type RM Length L Ch R = 1 ,34264   ,499,499,499
BEGIN DESCRIPTION:
UNT 020 IN LACR 60.0
END DESCRIPTION:
XS GIS Cut Line= 3
      2172406.88      13194735.9      2172997.17     13193235.87
      2172941.61     13192833.08
#Sta/Elev= 30
  3827.9  489.77  3913.7  487.88  4094.9  481.71  4144.1  479.41  4276.8  475.18
  4360.8  470.76  4385.2  470.86  4428.7  468.25  4493.2  466.64  4577.5  468.51
    4637  467.69  4654.4  468.72  4745.4  468.82  4769.8  467.97  4820.8  467.85
  4883.5  466.99  4913.3   467.4  4959.1  463.25  4961.8  462.75  4965.1  463.25
  4967.4  464.51  5016.2  468.15  5021.6  468.97  5037.4  469.07  5316.9  476.93
  5441.9  479.09  5529.8  482.84    5677  487.13  5697.6  487.83  5846.5  491.11
#Mann= 9 ,-1 , 0
  3827.9      .1       0  3913.7     .05       0  4094.9      .1       0
  4820.8     .12       0  4959.1     .07       0  4965.1     .12       0
  5037.4      .1       0    5677     .05       0  5697.6      .1       0
#XS Ineff= 2 , 0
         4654.83  468.72
Permanent Ineff=
       F       F
Bank Sta=4428.7,5016.2
XS Rating Curve= 0 ,0
Exp/Cntr=0.3,0.1

Type RM Length L Ch R = 1 ,33765   ,499,499,499
BEGIN DESCRIPTION:
UNT 020 IN LACR 59.0
END DESCRIPTION:
XS GIS Cut Line= 3
      2173011.06     13194659.48      2173274.95     13193603.92
      2173233.28     13192965.03
#Sta/Elev= 30
  4213.9  487.91  4283.2  485.89  4443.4  480.22  4628.4  470.96  4659.8   470.7
  4742.3   466.4  4804.2  465.26  4845.4  464.18  4896.9  466.04  4922.2  465.93
    4933  465.02  4948.5  464.71  4963.4  462.87  4969.1  460.66  4976.4  459.88
  4979.1  459.38  4982.4  459.88  4999.5  463.58  5012.6  464.45  5061.8  465.27
  5103.1  466.76  5210.8   467.5  5293.3  469.74  5340.1  469.78  5509.5  472.98
  5669.8  477.07  5689.8  476.88  5729.9  478.33    5760  478.04  5942.2  482.09
#Mann= 6 ,-1 , 0
  4213.9     .05       0  4283.2      .1       0    4933     .12       0
  4976.4     .07       0  4982.4     .12       0  5012.6      .1       0
#XS Ineff= 2 , 0
         4895.45  466.04
Permanent Ineff=
       F       F
Bank Sta=4804.2,5061.8
XS Rating Curve= 0 ,0
Exp/Cntr=0.3,0.1

Type RM Length L Ch R = 1 ,33266   ,632,632,632
BEGIN DESCRIPTION:
UNT 020 IN LACR 58.0
END DESCRIPTION:
XS GIS Cut Line= 3
       2173254.1      13194659.5      2173962.45     13193041.42
      2174149.42     13192570.51
#Sta/Elev= 30
  4112.9  479.87  4177.9  479.45    4180  479.43  4563.6  466.38  4727.1  465.86
  4779.5  464.86  4792.6  462.77  4814.4  464.18  4883.9  461.95  4959.5  463.05
    4997  457.05  4999.8  456.55    5003  457.05  5043.7   462.4  5152.1   466.5
  5227.7  466.22  5256.5   463.4  5279.9   466.4  5332.1  465.01  5371.2  468.54
  5576.9  471.04  5605.7  474.05  5611.3  478.27  5629.1  471.44  5704.7   469.5
  5742.3  472.63    5757  478.56  6011.7   478.2  6056.3  483.01  6385.9  496.31
#Mann= 6 ,-1 , 0
  4112.9     .05       0  4177.9      .1       0    4180     .16       0
    4997     .07       0    5003     .16       0  6385.9     .05       0
#XS Ineff= 1 ,-1
 4723.01 4907.67  463.77
Permanent Ineff=
       F
Bank Sta=4959.5,5043.7
XS Rating Curve= 0 ,0
Exp/Cntr=0.3,0.1

Type RM Length L Ch R = 1 ,32634   ,337,337,337
BEGIN DESCRIPTION:
UNT 020 IN LACR 57.0
END DESCRIPTION:
XS GIS Cut Line= 3
      2173487.75     13194646.83      2174037.72     13194196.85
      2174037.72     13193396.85
#Sta/Elev= 30
  4289.4  475.68  4346.1  473.07  4374.8  472.72  4417.9  470.78  4424.3  471.17
  4431.5  470.33  4445.1  470.83  4523.4  468.85  4630.3  464.91    4659  465.18
  4687.8  464.11  4829.9  462.67  4915.4  460.67  4986.4  457.39  4992.8  455.39
  5002.5  455.33    5007  454.34  5009.8  453.84    5013  454.34    5030  457.48
    5060  458.62    5100  458.71    5120  460.75  5143.3  461.56    5230  462.95
    5270  462.44    5510  466.99    5720  468.85    5790  470.21    5800  471.14
#Mann= 5 ,-1 , 0
  4289.4     .16       0  4915.4     .16       0    5007     .07       0
    5013     .16       0  5143.3      .1       0
#XS Ineff= 2 , 0
       0                    5230       0  462.95
Permanent Ineff=
       F       T
Bank Sta=4986.4,5030
XS Rating Curve= 0 ,0
Exp/Cntr=0.3,0.1

Type RM Length L Ch R = 1 ,32297   ,619,619,619
BEGIN DESCRIPTION:
UNT 020 IN LACR 56.0
END DESCRIPTION:
XS GIS Cut Line= 3
      2173517.99     13195340.04      2174122.17      13194819.2
      2174559.66      13193735.9
#Sta/Elev= 30
  3692.9  480.52  3843.8  477.78    4241  465.26  4361.6  462.94  4479.8  462.08
    4514  462.33    4531  461.68  4692.7  460.48  4884.8  460.53  4913.7  459.93
  4924.6  460.46  4978.4  456.62  5002.4  456.31  5018.2  453.35  5020.9  452.85
  5024.2  453.35  5032.4  455.41  5043.1  455.93  5056.1  455.77  5074.8  456.79
  5080.2  455.47  5118.6  456.72    5151  459.47    5158  459.34  5163.4  457.78
  5211.7  460.63  5280.4  460.64  5378.1   461.8  5526.8  461.84  5658.9  461.84
#Mann= 9 ,-1 , 0
  3692.9     .05       0  4479.8      .1       0    4531     .05       0
  4692.7      .1       0  4884.8     .16       0  5018.2     .07       0
  5024.2     .16       0  5280.4     .05       0  5526.8      .1       0
Bank Sta=5002.4,5043.1
XS Rating Curve= 0 ,0
Exp/Cntr=0.3,0.1

Type RM Length L Ch R = 1 ,31678   ,379,379,379
BEGIN DESCRIPTION:
UNT 020 IN LACR 55.0
END DESCRIPTION:
XS GIS Cut Line= 4
      2173636.09     13195742.79      2174733.28     13194805.31
       2174955.5     13194166.42      2174886.06     13193263.68
#Sta/Elev= 30
  3232.5  475.75  3386.9  471.49  3493.4  469.36    3500  469.91    3765  463.87
  3938.5  461.73  4025.4  460.85  4554.6  458.27    4889  456.35  4914.9   450.1
  4928.1  448.53  5020.4  448.48  5023.2  447.98  5026.4  448.48  5042.5  448.72
  5055.2  448.68  5061.4  449.84  5096.2  455.22  5101.5  454.71  5108.1  455.58
  5139.9  457.07  5266.5  459.44  5371.7  462.66  5441.9  463.42  5632.5   460.9
  5772.9  460.34  6003.6  462.28  6096.1   465.1  6103.9  464.58  6257.5  467.44
#Mann= 11 ,-1 , 0
  3232.5      .1       0    3765     .05       0  3938.5      .1       0
  4025.4     .05       0  4554.6      .1       0  5020.4     .07       0
  5026.4      .1       0  5042.5     .12       0  5061.4      .1       0
  5266.5     .05       0  6096.1      .1       0
Bank Sta=4889,5108.1
XS Rating Curve= 0 ,0
Exp/Cntr=0.3,0.1

Type RM Length L Ch R = 1 ,31299   ,624,624,624
BEGIN DESCRIPTION:
UNT 020 IN LACR 54.0
END DESCRIPTION:
XS GIS Cut Line= 4
      2174830.51     13196583.06        2175018.      13194944.2
      2175136.06     13194353.92      2175108.32     13193050.13
#Sta/Elev= 30
  3149.2  475.96  3507.7  468.54  3537.9  470.17  3558.1  467.54  3768.5  461.42
  3910.3  459.32  3950.6  456.76  3990.9   459.3  4232.4  459.42  4483.7  457.97
  4524.3  456.43  4667.3  454.97  4695.4  454.17  4793.5  456.18  4857.2  456.59
    4997  451.61  4999.7  451.11    5003  451.61  5061.2  454.95  5122.4  460.21
  5193.8  463.01  5235.2  462.89  5316.1  458.27  5367.1  457.29  5667.8  462.41
  5988.1   459.3    6087  460.22  6284.8  461.46    6448  464.24  6704.8  472.27
#Mann= 8 ,-1 , 0
  3149.2     .05       0  3768.5      .1       0  4793.5     .05       0
    4997     .03       0    5003     .05       0  5988.1      .1       0
    6087     .05       0  6284.8      .1       0
#XS Ineff= 2 , 0
         4822.73  456.57
Permanent Ineff=
       F       F
Bank Sta=4667.3,5061.2
XS Rating Curve= 0 ,0
Exp/Cntr=0.3,0.1

Type RM Length L Ch R = 1 ,30675   ,933,933,933
BEGIN DESCRIPTION:
UNT 020 IN LACR 53.0
END DESCRIPTION:
XS GIS Cut Line= 3
      2175011.07     13196423.34      2175545.78     13195298.37
      2175795.78     13193103.94
#Sta/Elev= 30
  3444.1  476.21  3611.4  472.02  3702.3  467.95  3707.8  468.88  3815.9  466.27
  3960.6  460.46  4138.8  456.03  4159.9  455.66  4502.2  454.63  4592.2  454.12
  4781.8  452.59  4886.2  452.27    4973  450.96  5009.1   446.1  5011.9   445.6
  5015.1   446.1  5023.3  448.73  5053.5  451.02    5124   452.4  5131.7  452.68
  5191.1  453.39  5726.3  452.21    5818  453.26  6058.7  455.64  6140.5  457.06
  6436.9   458.7  6523.8  459.93  6583.5  460.49  6781.3  463.02  6898.3  463.38
#Mann= 16 ,-1 , 0
  3444.1     .05       0  3960.6      .1       0  4138.8     .05       0
  4159.9      .1       0  4502.2     .05       0  4592.2      .1       0
  4886.2     .12       0  5009.1     .07       0  5015.1     .12       0
  5131.7     .12       0  5726.3      .1       0    5818     .05       0
  6058.7      .1       0  6436.9     .05       0  6523.8      .1       0
  6583.5     .12       0
#XS Ineff= 2 , 0
                         5191.15           453.4
Permanent Ineff=
       F       F
Bank Sta=4781.8,5124
XS Rating Curve= 0 ,0
Exp/Cntr=0.3,0.1

Type RM Length L Ch R = 1 ,29742   ,470,470,470
BEGIN DESCRIPTION:
UNT 020 IN LACR 52.0
END DESCRIPTION:
XS GIS Cut Line= 3
      2175511.03     13196124.78      2176295.78     13195235.87
        2176983.     13193472.71
#Sta/Elev= 30
  3450.4  460.09  3491.1  458.83  3722.9  454.43  3886.1  452.07  4059.1  451.72
  4207.1  450.73  4509.4  452.26  4806.8  450.23  4821.7  451.07    4839  449.62
  4930.4  446.27  4946.3  446.84  4960.3  445.88  4978.3  441.59  4981.5  442.09
  4984.8  447.09  4990.2  446.32  5063.7  449.78  5171.7  450.17  5332.7  447.72
  5434.7  448.55    5504  448.35  5676.8  450.87  6019.6  460.05  6169.3  465.51
  6266.5  469.16  6311.1   472.5  6352.3  472.95  6419.8   477.7  6528.5  482.51
#Mann= 10 ,-1 , 0
  3450.4     .05       0  3491.1      .1       0  3722.9      .1       0
  4059.1      .1       0  4207.1      .1       0  4821.7     .07       0
  5063.7      .1       0  5434.7     .12       0  5676.8      .1       0
  6169.3     .05       0
#XS Ineff= 2 , 0
       0 4558.58  452.31 5123.48       0  450.36
Permanent Ineff=
       T       T
Bank Sta=4839,5063.7
XS Rating Curve= 0 ,0
Exp/Cntr=0.3,0.1

Type RM Length L Ch R = 1 ,29272   ,526,526,526
BEGIN DESCRIPTION:
UNT 020 IN LACR 50.0
END DESCRIPTION:
XS GIS Cut Line= 3
      2175969.41     13196194.18      2176622.17      13195319.2
      2177323.12     13194354.52
#Sta/Elev= 30
  3509.9  459.18  3626.3     457  3735.1  455.22  3764.3   453.6    3879  452.62
  3899.8  451.56  4014.5  449.27  4142.9  447.99  4215.6  448.79  4414.8  452.18
  4599.9  453.05  4721.7  451.92  4814.6  449.28  4836.9  448.01  4843.1  448.53
  4857.8  447.53  4937.4  445.13  4993.8   445.8  5022.9  441.93  5037.1  445.16
  5064.9  448.02  5101.7  448.27  5107.4  448.06  5222.5   445.6    5245  443.78
  5280.5  444.33  5316.1   446.2  5381.3  447.21  5573.5  451.07    5794  460.14
#Mann= 8 ,-1 , 0
  3509.9     .05       0  3626.3      .1       0  4215.6      .1       0
  4857.8     .07       0  5064.9     .12       0  5101.7      .1       0
  5107.4     .12       0  5381.3      .1       0
#XS Ineff= 2 , 0
       0 4601.48  453.08 5100.85       0  448.29
Permanent Ineff=
       T       T
Bank Sta=4857.8,5064.9
XS Rating Curve= 0 ,0
Exp/Cntr=0.3,0.1

Type RM Length L Ch R = 1 ,28746   ,337,337,337
BEGIN DESCRIPTION:
UNT 020 IN LACR 49.0
END DESCRIPTION:
XS GIS Cut Line= 2
      2176830.52     13196409.44      2177559.42     13194521.24
#Sta/Elev= 30
  3753.8  466.04  4118.3  452.09  4287.3  448.25  4490.6  446.27  4511.8  446.16
  4614.1  446.48    4657  445.52  4784.5   443.2  4819.1   443.9  4914.2  444.88
  4982.8  443.36  4989.3  442.59    4997  440.15  4999.7  439.65    5003  440.15
  5021.4  443.98  5037.4  443.13    5075  444.28  5107.2   443.9  5139.3  442.96
  5151.9  441.46  5160.8  443.17  5225.1  445.46  5225.5  445.46  5278.7  446.68
  5463.4  454.73  5623.7  462.03  5664.6  462.89  5676.5  464.62  5777.8  467.62
#Mann= 10 ,-1 , 0
  3753.8     .05       0  4490.6      .1       0  4511.8     .12       0
  4784.5      .1       0  4819.1     .12       0    4997     .07       0
    5003     .12       0  5225.5      .1       0  5463.4     .05       0
  5676.5      .1       0
#XS Ineff= 2 ,-1
 4620.74  4860.8   444.9  5076.7  5777.8  444.33
Permanent Ineff=
       F       F
Bank Sta=4657,5225.1
XS Rating Curve= 0 ,0
Exp/Cntr=0.3,0.1

Type RM Length L Ch R = 1 ,28409   ,442,442,442
BEGIN DESCRIPTION:
UNT 020 IN LACR 48.0
END DESCRIPTION:
XS GIS Cut Line= 2
      2177233.28     13196409.49      2177760.85     13194771.24
#Sta/Elev= 30
  3873.9  464.05  3924.7  462.86  3960.7  460.42    3968  459.28  3973.2  460.19
  4139.3  453.69  4232.8  450.96  4380.9  447.35  4601.6  444.54  4689.4  442.62
  4716.1  442.25  4843.2  444.09  4881.7  443.34  4913.8  443.64  4951.1  442.57
  4990.3  443.04  5000.8  441.88  5012.2  439.25    5015  438.75  5018.2  439.25
  5021.8  440.41  5032.3  441.04  5072.2  442.48  5095.3  444.36  5137.4  445.57
  5143.5  446.52  5148.7  446.33  5180.8  448.61  5342.6  455.15    5595  464.69
#Mann= 8 ,-1 , 0
  3873.9      .1       0  3924.7     .05       0  4232.8      .1       0
  4689.4     .12       0  5012.2     .07       0  5018.2     .12       0
  5072.2      .1       0  5342.6     .05       0
#XS Ineff= 2 , 0
          4844.2  444.09
Permanent Ineff=
       F       F
Bank Sta=4601.6,5095.3
XS Rating Curve= 0 ,0
Exp/Cntr=0.3,0.1

Type RM Length L Ch R = 1 ,27967   ,496,496,496
BEGIN DESCRIPTION:
UNT 020 IN LACR 47.0
END DESCRIPTION:
XS GIS Cut Line= 3
      2177684.67     13196458.07      2177983.28     13195263.64
       2177830.5     13194826.14
#Sta/Elev= 30
  4009.2  468.84    4163   459.6  4329.1  451.57  4474.3  445.64  4525.8  445.27
  4567.1  443.94  4628.9  443.06  4680.5  442.87  4852.4  440.83  4896.9  439.39
  4958.8  441.07  4969.1  440.75  4984.6   436.8  4987.4   436.3  4990.6   436.8
    5000  440.59    5034  441.21  5061.8  442.76  5072.6  443.15  5082.5     443
  5123.7  445.03  5157.7  445.03  5193.8  446.15  5247.6  446.74  5424.3  452.66
  5485.3  454.12  5586.5  458.31  5650.1   459.9  5666.4  461.08  5703.8  462.11
#Mann= 7 ,-1 , 0
  4009.2     .05       0  4329.1      .1       0  4852.4     .12       0
  4984.6     .07       0  4990.6     .12       0  5072.6      .1       0
  5424.3     .05       0
#XS Ineff= 2 , 0
          4958.3  441.18
Permanent Ineff=
       F       F
Bank Sta=4680.5,5061.8
XS Rating Curve= 0 ,0
Exp/Cntr=0.3,0.1

Type RM Length L Ch R = 1 ,27471   ,482,482,482
BEGIN DESCRIPTION:
UNT 020 IN LACR 46.0
END DESCRIPTION:
XS GIS Cut Line= 3
      2177537.74     13196696.84      2178337.72     13195696.85
      2179537.73     13194596.84
#Sta/Elev= 30
  3719.4   480.1    3797  478.81    3805  477.74  3897.9  474.49  4110.8  463.52
  4160.4  462.05  4189.2  459.88  4363.7  452.34  4544.6  447.03  4615.8  443.98
  4743.9  441.54  4853.2  440.43  4978.4  438.76  4983.4  435.99  4986.1  435.49
  4989.4  435.99  4996.8  438.66  5013.9  439.68  5087.2  439.84  5122.1  440.41
  5226.6  440.85  5261.8  437.74  5283.3  440.38  5290.1  439.73  5325.6  441.53
  5495.8   445.7  5764.3  452.06  6111.5  455.26    6437  463.41  6627.9   469.5
#Mann= 8 ,-1 , 0
  3719.4     .05       0  4363.7      .1       0  4853.2     .12       0
  4983.4     .07       0  4989.4     .12       0  5087.2      .1       0
  5122.1     .12       0  5495.8      .1       0
#XS Ineff= 2 , 0
                         5224.15          440.89
Permanent Ineff=
       F       F
Bank Sta=4743.9,5325.6
XS Rating Curve= 0 ,0
Exp/Cntr=0.3,0.1

Type RM Length L Ch R = 1 ,26989   ,495,495,495
BEGIN DESCRIPTION:
UNT 020 IN LACR 45.0
END DESCRIPTION:
XS GIS Cut Line= 3
      2178087.75     13196596.82      2178637.72     13195996.85
      2179837.68     13194996.89
#Sta/Elev= 30
  4186.1  464.15  4525.5  452.12  4547.1  452.23  4709.9  445.86  4716.7  446.23
  4759.2  443.76  4858.5  440.27  4943.6  437.59  4968.9  434.56  4971.7  434.06
  4974.9  434.56  4978.7  436.55  4986.1  438.07  5014.2  438.59  5071.9  437.75
  5134.7  439.38  5276.6  440.23  5440.6  441.44  5689.3  445.03  5773.9  447.82
  5831.1  448.33  5937.2  451.88    5973  451.97  6057.6  455.66  6114.9   455.6
  6143.6  457.38  6262.2  461.42  6477.4  466.91  6534.1  469.62    6562  469.59
#Mann= 7 ,-1 , 0
  4186.1      .1       0  4968.9     .07       0  4974.9      .1       0
  5014.2     .12       0  5071.9      .1       0  6262.2     .05       0
  6477.4      .1       0
Bank Sta=4858.5,5276.6
XS Rating Curve= 0 ,0
Exp/Cntr=0.3,0.1

Type RM Length L Ch R = 1 ,26494   ,404,404,404
BEGIN DESCRIPTION:
UNT 020 IN LACR 44.0
END DESCRIPTION:
XS GIS Cut Line= 3
      2178387.73     13196746.85      2178987.72     13196346.85
      2180187.76     13196246.85
#Sta/Elev= 30
  4278.9  459.45  4502.7  450.77  4567.3  448.64  4574.8  449.14  4631.9  446.64
    4662  446.56  4706.6  444.48  4884.3  438.81  4931.9  437.11  4963.9   436.6
  4985.8  437.47  5002.5  437.02  5017.1  433.13  5019.8  432.63  5023.1  433.13
  5030.1  433.43  5042.9  436.12  5050.2  436.87  5100.3  435.54  5176.2  437.34
    5291  438.81  5366.1  441.65  5536.5  448.37  5561.9  448.42    5592   450.8
  5635.3  452.23  5780.2  454.75  5806.6  454.09  5973.4  457.58  6204.2  466.37
#Mann= 12 ,-1 , 0
  4278.9     .05       0  4706.6      .1       0  4931.9     .12       0
  4985.8     .16       0  5017.1     .07       0  5023.1     .16       0
  5042.9     .12       0  5176.2      .1       0  5366.1     .05       0
  5536.5     .08       0  5635.3     .05       0  5806.6      .1       0
Bank Sta=4884.3,5291
XS Rating Curve= 0 ,0
Exp/Cntr=0.3,0.1

Type RM Length L Ch R = 1 ,26090   ,200,200,200
BEGIN DESCRIPTION:
UNT 020 IN LACR 43.0
END DESCRIPTION:
XS GIS Cut Line= 4
      2178490.72     13196804.75      2178914.44     13196677.22
      2179480.31     13196535.65        2179897.     13196535.65
#Sta/Elev= 30
  4275.8  455.96  4377.1  451.71  4418.9  450.61  4439.8  449.11    4780  438.73
  4876.3   436.8  4886.6  435.25  4896.9   432.7  4903.6  429.68  4927.8  425.81
    4950  423.31  4966.1  422.97  4968.8  422.47  4972.1  422.97  4991.2  423.45
  5041.2  427.07  5051.5  428.43  5061.8  430.62  5068.5  433.06  5082.5  435.67
  5098.5  436.35    5113  437.05  5150.9  438.91  5257.7  443.51  5336.7  447.75
    5359  449.02    5389  449.59  5434.8  453.43    5559  459.59  5718.3  463.52
#Mann= 7 ,-1 , 0
  4275.8     .05       0  4966.1     .03       0  4972.1     .05       0
  5098.5      .1       0    5113     .05       0  5336.7     .08       0
  5434.8     .05       0
Bank Sta=4780,5150.9
XS Rating Curve= 0 ,0
Exp/Cntr=0.3,0.1

Type RM Length L Ch R = 1 ,25890   ,269,269,269
BEGIN DESCRIPTION:
Mapping XS 2ed1d341
END DESCRIPTION:
XS GIS Cut Line= 3
      2178473.38     13196908.91      2178985.52     13196856.83
      2179870.96     13196648.49
#Sta/Elev= 30
  4277.5  456.08  4347.2  452.68  4352.2  453.12  4412.5  450.89  4452.7  447.89
  4546.6  446.07  4593.5  443.33  4646.3  442.71    4796  438.32    4884  435.66
  4886.7  435.16    4890  435.66  4907.5     436  4928.1  438.89  4944.2  441.97
    5000  443.81  5020.5  443.41  5082.2  444.71  5133.6  444.17  5166.4   443.2
  5203.6  439.46    5226  439.75  5287.6  442.43  5298.7  443.72  5330.5  444.63
  5410.9  448.17    5432  450.12  5611.1  459.99  5685.2   463.4  5701.9  463.46
#Mann= 6 ,-1 , 0
  4277.5     .05       0    4884     .03       0    4890     .05       0
  5330.5     .08       0    5432     .05       0  5611.1      .1       0
Bank Sta=4796,4928.1
XS Rating Curve= 0 ,0
Exp/Cntr=0.3,0.1

Type RM Length L Ch R = 1 ,25621   ,552,552,552
BEGIN DESCRIPTION:
UNT 020 IN LACR 42.0
END DESCRIPTION:
XS GIS Cut Line= 4
      2178221.62     13197186.69      2178970.81     13197128.78
       2179619.2     13196978.36      2179983.25     13196752.99
#Sta/Elev= 30
  4025.9  464.01    4218  455.59  4348.1  450.69  4784.4  437.54    4809   437.8
  4835.8  436.42  4887.1  434.71  4894.3  434.67  4899.5  435.37  4928.1  434.44
  4943.5  434.77  4979.5  434.73    4997  432.49  4999.7  431.99    5003  432.49
  5020.5  434.88  5051.3  434.16    5098  434.72  5227.4  436.09  5245.9   436.7
  5384.1  442.58    5463  446.83  5487.8  448.16  5493.7   449.1  5509.1  448.81
  5537.8  450.49  5603.6  453.11  5661.5  456.28  5793.7  461.09  5871.1  464.38
#Mann= 9 ,-1 , 0
  4025.9      .1       0  4943.5     .12       0    4997     .07       0
    5003     .12       0    5098      .1       0  5227.4     .05       0
    5463     .08       0  5537.8     .05       0  5793.7      .1       0
Bank Sta=4835.8,5245.9
XS Rating Curve= 0 ,0
Exp/Cntr=0.3,0.1

Type RM Length L Ch R = 1 ,25069   ,482,482,482
BEGIN DESCRIPTION:
UNT 020 IN LACR 41.0
END DESCRIPTION:
XS GIS Cut Line= 3
      2178287.67     13197646.86      2179487.72     13197446.85
       2180087.7     13196846.87
#Sta/Elev= 30
  3783.4   464.3    3824   463.2  4039.7  454.32  4115.5  450.92  4120.5   451.2
  4181.4  449.06  4286.1  444.35  4480.4  437.62  4600.2   436.4  4700.2  435.83
  4784.6  435.28  4817.5  434.45  4888.5  432.51  4913.1  432.59  4949.3  432.73
  4994.5  429.81  4997.2  429.31  5000.5  429.81  5003.5  429.81  5014.1  431.86
  5078.8  432.86  5127.3  433.45  5169.7  434.74  5212.1  435.84    5263  438.18
  5286.5  439.34  5392.4   444.7  5755.6  460.56  5806.1  462.58  5848.5  465.34
#Mann= 13 ,-1 , 0
  3783.4     .05       0  4039.7      .1       0  4286.1     .05       0
  4600.2      .1       0  4700.2     .05       0  4913.1     .12       0
  4994.5     .07       0  5000.5     .12       0  5078.8      .1       0
    5263     .05       0  5286.5      .1       0  5392.4     .05       0
  5755.6      .1       0
Bank Sta=4817.5,5169.7
XS Rating Curve= 0 ,0
Exp/Cntr=0.3,0.1

Type RM Length L Ch R = 1 ,24587   ,463,463,463
BEGIN DESCRIPTION:
UNT 020 IN LACR 40.0
END DESCRIPTION:
XS GIS Cut Line= 3
      2178537.74     13198596.84      2179737.72     13197796.85
      2180037.76     13197596.83
#Sta/Elev= 30
  3557.8  462.25  3571.3  462.47  3580.3  461.71  3673.5  459.84  3802.7  454.76
  3817.7  453.59  3853.7  452.34  3868.8  450.97  3968.6  446.46  4199.3  438.45
  4379.5  435.37  4549.8  433.96  4740.1  433.04  4819.7  431.69  4884.3  431.92
  4950.4  430.77  4992.5  431.89    5003  431.22  5004.5  429.58  5007.3  429.08
  5010.5  429.58  5013.5  430.17  5028.5  430.49  5036.1  431.97  5064.6  432.92
  5072.1  433.93  5136.7  437.99  5202.8  443.95  5280.9   448.1  5360.6   451.4
#Mann= 7 ,-1 , 0
  3557.8     .05       0  3968.6      .1       0  4199.3     .05       0
  4379.5      .1       0  4549.8     .05       0  5004.5     .03       0
  5010.5     .05       0
Bank Sta=4740.1,5072.1
XS Rating Curve= 0 ,0
Exp/Cntr=0.3,0.1

Type RM Length L Ch R = 1 ,24124   ,491,491,491
BEGIN DESCRIPTION:
UNT 020 IN LACR 39.0
END DESCRIPTION:
XS GIS Cut Line= 3
      2178687.75     13198596.84      2179687.72     13198196.85
      2180237.72     13197696.86
#Sta/Elev= 30
    3923  459.79  4009.1  456.65  4093.9  452.48  4099.3  453.17  4116.8  451.59
    4207  448.06  4236.7  446.08  4255.5  446.02  4260.9  445.14  4278.4  445.52
  4290.5  444.49  4436.6   440.1  4505.9  437.25  4543.6  436.77  4676.9  433.13
    4829  431.41  5010.9  429.42  5013.6  428.92  5016.9  429.42  5100.1  429.97
  5172.4  431.16  5176.7  431.26  5361.2   437.9  5566.6  446.76  5587.5  447.32
  5601.7   446.6  5636.9  448.46  5665.3  448.94  5686.9  448.31  5743.3  450.31
#Mann= 7 ,-1 , 0
    3923     .05       0  4436.6     .08       0  4543.6     .05       0
  5010.9     .03       0  5016.9     .05       0  5100.1      .1       0
  5172.4     .05       0
Bank Sta=4829,5176.7
XS Rating Curve= 0 ,0
Exp/Cntr=0.3,0.1

Type RM Length L Ch R = 1 ,23633   ,491,491,491
BEGIN DESCRIPTION:
UNT 020 IN LACR 38.0
END DESCRIPTION:
XS GIS Cut Line= 3
      2179187.72     13198646.85      2179787.72     13198646.85
      2180387.74     13198596.85
#Sta/Elev= 30
    4400  443.22    4520  439.38    4550  437.84  4565.9  437.79  4664.1  435.59
    4700  435.33    4770  433.48    4870  429.87  4958.5  428.47    4960  428.46
    4970  427.01    4980  424.01    4987  419.95  4989.7  419.45    4993  419.95
  4997.5  421.08  5002.5  421.08    5010  424.12  5040.1  428.89    5057  429.19
  5090.3  429.18  5230.8  432.53  5260.9  432.36  5321.1  435.13  5341.2  435.08
  5441.5   439.3  5456.7  439.46  5511.8  442.21    5582  444.56  5602.1  445.88
#Mann= 8 ,-1 , 0
    4400     .05       0  4565.9     .08       0  4664.1     .05       0
  4958.5     .12       0    4987     .07       0    4993     .12       0
    5057      .1       0  5456.7     .05       0
Bank Sta=4960,5040.1
XS Rating Curve= 0 ,0
Exp/Cntr=0.3,0.1

Type RM Length L Ch R = 1 ,23142   ,298,298,298
BEGIN DESCRIPTION:
UNT 020 IN LACR 37.0
END DESCRIPTION:
XS GIS Cut Line= 3
      2179287.74     13198796.86      2179887.72     13199096.85
       2180487.7     13198796.86
#Sta/Elev= 30
  4329.2  439.32  4418.6  436.66  4463.3  436.76    4613  433.32  4835.1  429.83
  4924.5   427.4  4941.3  426.36  4946.9  426.87  4955.3  424.75  4963.7  421.49
  4969.3  426.88    4986  418.36  4988.6  418.27  4991.4  417.77  4994.6  418.27
  5022.4  420.28  5044.7  427.23  5060.7  426.62  5104.8  427.45  5304.7  432.02
  5343.8  433.69  5371.7   433.7  5402.5     436  5410.9  435.59  5447.2   437.3
  5467.4  437.39  5536.7  441.69  5626.1  446.09  5634.5  447.23  5670.8  448.48
#Mann= 7 ,-1 , 0
  4329.2     .05       0    4613      .1       0  4988.6     .07       0
  4994.6      .1       0  5060.7     .16       0  5104.8      .1       0
  5467.4     .05       0
Bank Sta=4946.9,5044.7
XS Rating Curve= 0 ,0
Exp/Cntr=0.3,0.1

Type RM Length L Ch R = 1 ,22844   ,474,474,474
BEGIN DESCRIPTION:
UNT 020 IN LACR 36.0
END DESCRIPTION:
XS GIS Cut Line= 3
      2179101.35     13199666.42      2180399.95     13199201.14
      2180747.21     13198992.79
#Sta/Elev= 30
  3978.7  447.65  4059.8  443.25  4313.9   435.4  4427.4  433.26  4498.4  432.78
  4532.8  430.79  4585.4  430.98  4638.2  428.94  4646.3  429.09  4686.5   426.9
  4703.1  428.57  4728.6  427.67  4743.6  428.83  4764.6  426.86    4814  427.86
  4907.8  426.79  4913.1  423.35  4930.9  418.67  4943.9  419.37  4954.4  417.78
  4959.7  417.13  4962.5  416.63  4965.7  417.13  4994.6  425.71  5112.4  427.95
  5281.4  432.32  5456.3  440.84  5491.2  443.07  5512.6  442.62  5763.1   457.5
#Mann= 11 ,-1 , 0
  3978.7      .1       0  4427.4     .05       0  4532.8      .1       0
  4638.2     .12       0  4646.3     .08       0  4743.6     .12       0
  4954.4     .16       0  4959.7     .07       0  4965.7     .16       0
  5112.4      .1       0  5456.3     .05       0
#XS Ineff= 2 , 0
         4740.06  429.15
Permanent Ineff=
       F       F
Bank Sta=4907.8,4994.6
XS Rating Curve= 0 ,0
Exp/Cntr=0.3,0.1

Type RM Length L Ch R = 1 ,22370   ,888,888,888
BEGIN DESCRIPTION:
UNT 020 IN LACR 35.0
END DESCRIPTION:
XS GIS Cut Line= 2
      2179587.46     13200270.57      2180691.64      13199353.9
#Sta/Elev= 30
  4130.8  441.68  4201.2  440.62  4261.1   439.7  4303.8  437.32  4318.1  437.11
    4326  438.48    4387  436.97  4410.6   437.2  4478.2  434.24    4645  428.78
  4792.8  426.56  4800.6  426.59  4931.4  424.96    4964  424.32  4986.1  415.71
  4997.5   414.1  5000.2   413.6  5003.5   414.1    5007  414.99  5014.8  419.87
  5021.7  420.85  5027.9  423.65  5035.6  424.66  5042.1  423.34  5070.8  423.94
  5099.4  425.91  5298.7  431.64  5354.6  432.26    5539  440.94  5565.9  441.33
#Mann= 11 ,-1 , 0
  4130.8      .1       0  4201.2     .08       0    4387      .1       0
  4478.2     .05       0  4792.8     .08       0  4800.6      .1       0
  4931.4     .12       0  4997.5     .07       0  5003.5     .12       0
  5021.7      .1       0    5539     .08       0
Bank Sta=4964,5027.9
XS Rating Curve= 0 ,0
Exp/Cntr=0.3,0.1

Type RM Length L Ch R = 1 ,21482   ,502,502,502
BEGIN DESCRIPTION:
UNT 020 IN LACR 34.0
END DESCRIPTION:
XS GIS Cut Line= 2
      2179955.52     13200756.69      2180969.38     13200006.71
#Sta/Elev= 30
  4462.4  443.34  4635.9  442.27  4739.6  437.06    4807  433.36  4864.4  428.85
  4913.4  426.88  4928.1  425.15  4950.2  420.21  4957.3  418.07  4989.3   415.9
  5007.4  413.41  5025.3  412.64    5028  412.14  5031.3  412.64  5036.7  415.52
  5042.9  415.05  5057.5  421.62  5099.5  423.98  5186.6  423.44  5245.6  425.01
  5322.6  425.84  5443.7  425.33  5514.6  426.42  5543.9  427.87  5564.7  427.61
  5579.4  425.92  5585.6  426.96  5657.3  427.53  5712.7  428.87  5723.5  429.06
#Mann= 9 ,-1 , 0
  4462.4      .1       0  4739.6     .08       0  4864.4      .1       0
  4989.3     .12       0  5025.3     .07       0  5031.3     .12       0
  5245.6      .1       0  5657.3     .05       0  5712.7      .1       0
Bank Sta=4950.2,5057.5
XS Rating Curve= 0 ,0
Exp/Cntr=0.3,0.1

Type RM Length L Ch R = 1 ,20980   ,523,523,523
BEGIN DESCRIPTION:
UNT 020 IN LACR 33.0
END DESCRIPTION:
XS GIS Cut Line= 3
      2180183.46     13201171.05      2180956.01     13200580.79
      2181954.28     13199530.43
#Sta/Elev= 30
  4365.4  439.25    4579  434.17  4589.2  433.98  4679.2  431.23  4913.9  424.89
  4949.7  423.97  4956.5  419.48  4962.8  418.33  4977.3  415.41    5000  414.02
  5017.9  408.53  5020.6  408.03  5023.9  408.53  5041.7  414.33  5048.6  414.41
  5070.8   417.5  5078.8   420.7  5113.3   421.2  5120.7  419.48    5156   416.5
  5163.6  418.62  5170.5  421.74  5234.9  423.45    5377   422.8    5667  427.06
    5973  433.64  6004.9  434.41  6155.2  438.43  6501.8  442.29  6786.7  450.61
#Mann= 11 ,-1 , 0
  4365.4      .1       0    4579     .05       0  4589.2     .08       0
  4679.2     .05       0  4913.9      .1       0  5017.9     .07       0
  5023.9      .1       0  5048.6     .12       0  5078.8      .1       0
    5973     .08       0  6004.9      .1       0
Bank Sta=4962.8,5163.6
XS Rating Curve= 0 ,0
Exp/Cntr=0.3,0.1

Type RM Length L Ch R = 1 ,20457   ,486,486,486
BEGIN DESCRIPTION:
UNT 020 IN LACR 32.0
END DESCRIPTION:
XS GIS Cut Line= 2
      2180531.93     13201492.78      2181600.76     13200611.34
#Sta/Elev= 30
  4252.9  438.97  4411.2  432.15  4450.2  430.81  4566.9  426.64  4620.2   425.7
  4694.5  425.35  4701.1  424.61  4843.7  421.81  4893.9  421.55  4943.4  420.28
  4949.9  419.88  4957.8  418.07  4978.6  412.43  4999.4   412.9  5013.7  411.17
  5025.1  408.74  5027.8  408.24  5031.1  408.74  5042.4  413.36  5050.3  414.15
  5055.5  415.76    5064  417.14  5078.7  419.09  5106.3  420.76  5134.9  420.71
  5209.9  423.13  5393.2  428.51  5400.2  428.89  5589.7  435.97  5638.3   436.8
#Mann= 11 ,-1 , 0
  4252.9     .05       0  4411.2     .08       0  4450.2     .05       0
  4620.2      .1       0  5025.1     .07       0  5031.1      .1       0
  5055.5     .12       0  5078.7      .1       0  5209.9     .05       0
  5393.2      .1       0  5400.2     .05       0
Bank Sta=4957.8,5064
XS Rating Curve= 0 ,0
Exp/Cntr=0.3,0.1
