HEC-RAS study NUECES RIVER.prj: NUECES RIVER Base Level Engineering

--- NUECES RIVER.g01 (geometry) --- (continued)

Type RM Length L Ch R = 1 ,310237  ,6332,6332,6332
BEGIN DESCRIPTION:
LOWER NUECES 40.0
END DESCRIPTION:
XS GIS Cut Line= 6
      2342448.39     13253484.62      2339661.35     13251908.57
      2331944.74     13251162.05      2327599.61     13248536.83
      2302128.33     13246382.15      2294067.41     13248381.65
#Sta/Elev= 30
-19587.8  226.16  -13328  208.13-9731.55  228.03-9012.25  193.76-8092.99   221.2
 -5744.6  190.67-4435.49  201.38-4355.55  171.26-4255.62  200.48-3196.21  190.63
-2716.35  161.77-2466.43  186.27 -2109.7  184.87 -1858.8  172.97 -1587.9  121.85
-1166.67   98.35    -986   90.71   13556   98.49 13877.4    95.5 14073.9   96.63
 14368.8    97.3 14750.3   99.55 19041.8   99.36   19872  123.83 19970.3  126.97
 22005.5  193.93 24288.5  213.17 25880.1  191.82 27613.9   223.7 30310.7  226.82
#Mann= 17 ,-1 , 0
-19587.8     .05       0 -9539.6      .1       0 -8470.1     .05       0
 -8365.1      .1       0 -8019.3     .05       0 -6779.5     .08       0
 -6666.8      .1       0 -2632.6      .1       0-1166.67    .033       0
 13286.3      .1       0 13877.4     .16       0 14073.9      .1       0
 14368.8     .16       0 14750.3     .05       0 19041.8      .1       0
   19872     .08       0 19970.3      .1       0
#XS Ineff= 1 ,-1
14730.2920580.91   98.06
Permanent Ineff=
       F
Bank Sta=-1166.67,13556
XS Rating Curve= 0 ,0
Exp/Cntr=0.3,0.1

Type RM Length L Ch R = 1 ,303905  ,4743,4743,4743
BEGIN DESCRIPTION:
LOWER NUECES 40.5
END DESCRIPTION:
XS GIS Cut Line= 4
      2338166.81     13250618.73      2324874.75     13243077.52
      2308273.19     13238628.74      2294384.26     13233149.12
#Sta/Elev= 30
-16427.9  219.65  -13934  221.59-13903.2  201.65-13838.3  196.96  -13578   199.2
  -13181  207.67-12958.6  206.16-11119.6  189.88 -9820.3  200.86-8221.08  154.76
-6701.82  156.25-5992.17  187.13-5532.39  188.97 -3762.9  149.43 -2673.3  124.43
 -1145.6  148.62  291.67   98.87   463.4   91.21   466.1   90.71   469.4   91.21
   570.5   91.2114041.67   98.87 14082.3  100.37 14384.8  102.52   14879  115.73
 15393.1  121.6216142.07  157.6816991.44  145.0917820.79  166.49 30972.5  193.13
#Mann= 20 ,-1 , 0
-16427.9     .05       0  -13578      .1       0  -13181     .05       0
-12958.6      .1       0-11344.9     .05       0-11024.4      .1       0
-10802.3     .05       0 -9803.1      .1       0 -3762.9      .1       0
   463.4    .033       0   469.4      .1       0   570.5    .033       0
 14082.3      .1       0 14384.8     .16       0   14879      .1       0
 15393.1      .1       0 17605.3     .05       0 18826.1      .1       0
 20934.7     .05       0 24425.3      .1       0
#XS Ineff= 1 ,-1
14232.3715103.73  108.51
Permanent Ineff=
       F
Bank Sta=291.67,14041.67
XS Rating Curve= 0 ,0
Exp/Cntr=0.3,0.1

Type RM Length L Ch R = 1 ,299162  ,6052,6052,6052
BEGIN DESCRIPTION:
LOWER NUECES 41.0
END DESCRIPTION:
XS GIS Cut Line= 5
      2340242.56     13249164.26      2329816.92      13240258.6
      2313453.59     13234972.51      2312446.04     13227531.62
      2302190.97     13222890.59
#Sta/Elev= 30
-20138.7  222.36-16119.4  198.82-15529.8  215.99-14330.6  184.27-14090.7  195.68
-13900.8  184.62-13001.4  187.24-12801.5  197.35-10722.8  161.12-9513.56  167.23
-8414.24  126.66-8094.43  132.91-7564.75  163.31-6785.23  139.15 -5285.7   139.2
 -4329.7  111.64 -3205.6  100.38-2386.31   99.03-2196.35   91.21    9750   98.35
 10657.1  136.6613700.75  145.8714330.75  135.3317680.75  166.4820020.07  148.93
21229.59  162.2924898.16  159.1526097.69  187.29 28128.8   185.9 29533.9  197.92
#Mann= 17 ,-1 , 0
-20138.7     .05       0-16248.3     .05       0  -13895     .05       0
-12792.3      .1       0-11050.3     .05       0-10126.1      .1       0
 -6990.8      .1       0 -4329.7      .1       0 -3205.6    .033       0
    9750     .05       0 10657.1      .1       0 11634.2      .1       0
 15998.6     .05       0 18260.6      .1       0 20295.6     .05       0
 26439.1      .1       0 28128.8      .1       0
Bank Sta=-2386.31,9750
XS Rating Curve= 0 ,0
Exp/Cntr=0.3,0.1

Type RM Length L Ch R = 1 ,293110  ,6526,6526,6526
BEGIN DESCRIPTION:
LOWER NUECES 42.0
END DESCRIPTION:
XS GIS Cut Line= 4
      2342276.45     13249742.15      2335218.69     13239762.82
       2313537.6     13227063.03       2303894.4     13222897.69
#Sta/Elev= 30
-24892.4  220.42-22380.8  215.11-17441.3  206.23-15282.6  165.06-14163.2  186.01
-12704.1  177.93-11114.3  154.07-10244.4  125.81-9634.46  128.33-8864.54  110.08
 -3564.5   98.88 -2669.7   94.17 -1663.2   92.79  -619.9   96.81   132.4   90.71
  9107.8   91.21  9173.4  100.14  9488.1  119.89  9515.4  107.669642.219  108.98
9842.219  132.3210082.22  111.1710362.22  132.3910682.22  105.9211622.22  158.44
18999.66  157.0620229.18  160.9421568.66  186.65   22771  168.65 22961.6  176.51
#Mann= 18 ,-1 , 0
-24892.4     .05       0-22380.8     .05       0-16257.4     .05       0
-15021.7     .05       0-13092.8      .1       0  -11980     .05       0
 -9715.9      .1       0   -8440      .1       0 -7147.8     .05       0
 -3564.5     .05       0 -2669.7     .05       0 -1663.2     .05       0
  -619.9    .033       0    9968     .08       0 12316.5      .1       0
 14869.7     .05       0 20175.2      .1       0 22563.2      .1       0
Bank Sta=-3564.5,9173.4
XS Rating Curve= 0 ,0
Exp/Cntr=0.3,0.1

Type RM Length L Ch R = 1 ,286584  ,5106,5106,5106
BEGIN DESCRIPTION:
LOWER NUECES 43.0
END DESCRIPTION:
XS GIS Cut Line= 4
      2346877.69     13247986.21      2335839.61     13231293.92
      2317828.97     13224392.37      2303414.98     13221721.64
#Sta/Elev= 30
-26467.8  197.97-21299.1  193.09-19889.7  167.18-18890.1  192.76-15681.3   198.4
-14541.8  183.24  -13992  141.34  -13852  143.06-13792.1  196.69-13642.1  198.22
-13592.1  152.16-13272.3  141.34-12322.6  139.47-11782.8  168.01-9093.94  106.59
-8044.35  128.76 -5921.6  105.08 -5358.3   97.16 -5331.3   91.14  8506.6   97.74
  9502.3  142.81 10662.7  129.66 12512.7  172.69 16472.7     151 18842.7  153.04
 20072.7  183.95 23062.7  154.74 26052.7  179.09 26722.7  156.18   27491  181.77
#Mann= 17 ,-1 , 0
-26467.8     .05       0-19373.7     .05       0-17924.3     .05       0
-14914.1     .05       0-12882.7     .05       0-11331.1     .05       0
 -8714.2     .05       0 -5921.6    .033       0  9714.2      .1       0
 11277.6     .05       0 14497.1     .05       0 18781.2      .1       0
 20112.9     .05       0 23294.7      .1       0   24127     .05       0
 25592.7      .1       0 26668.7      .1       0
Bank Sta=-5358.3,8506.6
XS Rating Curve= 0 ,0
Exp/Cntr=0.3,0.1

Type RM Length L Ch R = 1 ,281478  ,3441,3441,3441
BEGIN DESCRIPTION:
LOWER NUECES 44.0
END DESCRIPTION:
XS GIS Cut Line= 4
      2348281.65     13232276.32      2337032.12     13221025.45
      2316709.11     13223170.42      2303280.84      13221493.9
#Sta/Elev= 30
-22332.1  165.88-20130.7   158.2-17040.3  140.63-16130.8  152.11-14072.1   141.3
-13932.2  126.68-13462.5  139.53-11213.8  113.36-10314.3  129.91-4696.99  132.79
   -3375   98.42 -3280.4   90.6410916.67   98.74 10928.3  120.67 10976.2  144.78
 11172.1  140.65 11250.1  108.68 11567.4  108.75 12028.2  109.85   12121  135.06
12549.73  161.4813569.58  174.5516128.68  144.1916868.39  164.5918527.74  154.77
19757.26  179.19   22966  154.6725984.82  171.13 26554.6  153.58 27546.5   178.7
#Mann= 18 ,-1 , 0
-22332.1     .05       0-20130.7     .05       0-18654.7     .05       0
-17845.4     .05       0-16994.5      .1       0-14660.8     .05       0
-13662.7     .05       0-10594.8     .05       0 -4958.7      .1       0
   -3375    .033       0 11567.4      .1       0 13904.1     .05       0
 18945.6      .1       0 20355.9     .05       0 22969.4      .1       0
 23985.6     .05       0   25041     .05       0 25762.3      .1       0
Bank Sta=-3375,10916.67
XS Rating Curve= 0 ,0
Exp/Cntr=0.3,0.1

Type RM Length L Ch R = 1 ,278037  ,7861,7861,7861
BEGIN DESCRIPTION:
LOWER NUECES 45.0
END DESCRIPTION:
XS GIS Cut Line= 5
      2352372.36     13237347.63      2339800.36     13219371.69
      2335902.84     13217478.39      2318391.49     13219792.72
      2303283.07     13220608.25
#Sta/Elev= 30
-32727.1  178.47-18089.7  148.25-15740.2  126.08-4768.63  130.92-3298.61   98.09
   -3195   90.64 9777.78   97.77  9837.6  134.69    9951  140.15 10039.3  140.07
 10150.3   99.27 10271.3  135.82   10352  132.02 10436.8  101.32 10466.2   110.5
 10553.7  142.31 10662.2  116.29 10740.7  138.06   11009  145.44 12280.9  107.21
 12648.9  122.39 14524.1  154.75 15641.5  138.73   16586   156.8 17628.7  167.42
 19058.3  138.58 20008.3  132.03 23045.7  149.44 25549.9  150.89   26336  164.69
#Mann= 17 ,-1 , 0
-32727.1     .05       0-23814.3     .05       0-22296.1     .05       0
-18932.6     .05       0-16489.3     .05       0-15354.3     .05       0
 -4257.9      .1       0-3298.61    .033       0    9951     .16       0
 10466.2      .1       0   11009     .05       0 12648.9     .05       0
   16586      .1       0 19058.3      .1       0 20008.3     .05       0
 23045.7     .05       0 25549.9      .1       0
Bank Sta=-3298.61,9777.78
XS Rating Curve= 0 ,0
Exp/Cntr=0.3,0.1

Type RM Length L Ch R = 1 ,270176  ,5572,5572,5572
BEGIN DESCRIPTION:
LOWER NUECES 46.0
END DESCRIPTION:
XS GIS Cut Line= 6
      2353562.71       13238190.      2346950.55     13226596.34
      2339491.07      13217915.3      2328062.94     13211351.23
      2306660.25     13210366.46      2300703.16     13210927.31
#Sta/Elev= 30
-37993.4  174.01-23570.9  160.34-18602.8  129.08 -634.96  131.25  1562.5   97.87
  1783.1   90.71 6881.87   98.35  6933.4  112.88  6993.4  102.79  7453.4  109.17
7745.949   124.9 8894.77  123.47 8934.77   132.69274.762  109.72 9474.75  124.22
 9544.75   139.1 9694.75  128.39 9834.75  142.4210744.72  155.79 12014.7  131.94
13684.66     188 16054.6  191.5616934.58  169.4618194.55  190.1318894.54  178.41
19624.52  197.25 20774.5  187.1923382.21  200.5424440.96   192.1 27399.5   214.7
#Mann= 17 ,-1 , 0
-37993.4     .05       0-27102.7     .05       0-25602.6     .05       0
-21631.9     .05       0-19140.8     .05       0   -5885      .1       0
 -4490.2     .05       0  1562.5    .033       0  6993.4      .1       0
  8237.7      .1       0    9109      .1       0 11012.5      .1       0
 17259.9     .05       0 19377.6      .1       0 22076.2     .16       0
 22833.3      .1       0 24069.3      .1       0
Bank Sta=1562.5,6881.87
XS Rating Curve= 0 ,0
Exp/Cntr=0.3,0.1

Type RM Length L Ch R = 1 ,264604  ,5507,5507,5507
BEGIN DESCRIPTION:
LOWER NUECES 47.0
END DESCRIPTION:
XS GIS Cut Line= 4
      2345545.36     13218554.98      2331764.94     13207758.51
      2324386.47     13206944.71      2306808.33      13206727.7
#Sta/Elev= 30
-17643.7  157.29-16752.5  140.62  -15917   131.1 -1322.2  132.34   565.3  129.38
  1019.7  115.07  2445.2  134.19  2555.9   129.9  2596.1   96.99  2603.2   91.21
  2609.2   91.21  6401.8   91.21  6439.3    96.9  6519.8  126.05  6710.9  106.77
  6962.4  143.46 9322.09  140.39 9882.09  164.8711922.09  137.6513192.09  154.36
14602.09  145.0515982.09  167.8717902.09  158.9919862.09  191.7921702.09  176.33
 22807.5  188.87 23248.8  188.26   24190  186.82   24850  190.54 24865.1  190.63
#Mann= 18 ,-1 , 0
-17643.7     .08       0-16752.5     .05       0  -15917     .05       0
 -1322.2     .16       0  2609.2    .033       0  6401.8      .1       0
   11322      .1       0 12113.3     .05       0 14278.3     .08       0
 15063.2     .05       0 17202.1     .05       0 17747.1      .1       0
 18522.5      .1       0 21927.7     .05       0 22807.5      .1       0
 23248.8     .05       0   24190      .1       0   24850     .05       0
Bank Sta=2596.1,6439.3
XS Rating Curve= 0 ,0
Exp/Cntr=0.3,0.1

Type RM Length L Ch R = 1 ,259097  ,3451,3451,3451
BEGIN DESCRIPTION:
LOWER NUECES 48.0
END DESCRIPTION:
XS GIS Cut Line= 4
      2345816.61     13217144.37       2333446.8     13207487.24
      2327044.89     13198752.44      2318255.82     13191265.45
#Sta/Elev= 30
-16273.8  133.19-16013.4  133.04-14517.7  134.67-13078.4  118.54-13038.4  124.97
-11399.1  127.36-54.0498  135.26745.9395  130.35  1286.3  100.82    1487   94.84
  1578.6   90.71  7088.7   91.21    7118  102.48 7118.06    95.9  7153.5  110.59
7675.939  141.988425.939  152.748955.939  149.759445.939  166.2410205.94  158.28
11305.53  163.5811915.29  153.1112734.97  165.0514404.32  163.0516033.69  174.61
16943.33  163.3418502.72  167.4819632.28  185.1520681.87  168.85 21794.6  172.03
#Mann= 18 ,-1 , 0
-16273.8     .05       0-16013.4      .1       0-13950.9     .05       0
 -8632.3      .1       0 -7671.9     .05       0 -5710.4     .05       0
 -1668.1     .16       0  -777.2     .16       0   656.6      .1       0
  1286.3    .033       0  7153.5      .1       0  8679.3      .1       0
  9477.4     .05       0   11622     .05       0   13312      .1       0
 14786.5      .1       0 15836.2      .1       0 17533.6     .05       0
Bank Sta=1487,7118.06
XS Rating Curve= 0 ,0
Exp/Cntr=0.3,0.1

Type RM Length L Ch R = 1 ,255646  ,507,507,507
BEGIN DESCRIPTION:
LOWER NUECES 49.0
END DESCRIPTION:
XS GIS Cut Line= 6
      2345209.73     13215688.79      2333079.98      13206557.3
      2333639.87     13202675.35      2331362.96     13197412.33
      2327184.12      13197854.8      2319429.52     13191601.09
#Sta/Elev= 30
  -16173  134.95-15781.8  134.77-13987.3  117.43-2148.84  136.42 -1598.9   124.5
-1180.31  135.33 -544.95  133.6274.37012  109.11  1112.8  114.79  1570.2   97.63
  1982.4   90.71 6339.29   98.01  6661.1   123.1  6952.7  112.64  7040.6  124.23
  7262.9  112.267659.881  132.78 8119.43  119.5610285.93  145.5111274.09  136.86
12212.33  159.6812980.96  146.6513550.51  156.8114060.11  141.2114879.47  158.95
16588.13  147.7618216.86  168.9519236.06  162.2722163.77  183.96   22887  176.69
#Mann= 18 ,-1 , 0
  -16173     .08       0-15781.8      .1       0-15049.9     .05       0
 -6219.8     .05       0 -3167.6     .16       0 -2066.9     .16       0
    -877      .1       0  1112.8     .05       0  1570.2    .033       0
 6339.29      .1       0    7899     .05       0 12256.3      .1       0
   12884     .05       0 13360.9      .1       0 13708.2     .05       0
 15500.9      .1       0 19576.9     .05       0 22170.6     .05       0
Bank Sta=1570.2,6339.29
XS Rating Curve= 0 ,0
Exp/Cntr=0.3,0.1

Type RM Length L Ch R = 1 ,255139  ,776,776,776
BEGIN DESCRIPTION:
LOWER NUECES 50.0
END DESCRIPTION:
XS GIS Cut Line= 6
      2345717.71     13215183.12      2333272.11     13206545.23
      2334331.91     13202546.87       2331528.2     13197340.28
      2327269.34     13197713.87      2320041.62     13191774.81
#Sta/Elev= 30
-16585.8  131.25-16322.7   130.2  -13687  116.55-12237.1  127.57-2217.32  139.17
-1567.32  119.13 -1436.7  132.01  -294.3  119.48   546.5  109.76   548.4     106
  3450.1     106  3455.8    94.3  4784.6    94.3  4800.8     106  5167.5     106
    5177    93.8  5632.4    93.8 5632.56     106    6859     106    7369  143.24
  7565.4  140.55 9285.58  122.36 10973.6  144.3611702.74  136.1712711.56  159.22
14390.22  138.4115209.74   151.616488.99  142.2318438.23  165.13 22346.7  182.44
#Mann= 17 ,-1 , 0
-16585.8     .08       0-16322.7     .05       0-13810.7     .05       0
 -4634.2     .05       0 -3697.4     .16       0 -2292.4     .16       0
 -1436.7      .1       0  -294.3      .1       0   546.5     .05       0
   548.4    .013       0    6859     .05       0    6859      .1       0
  7565.4     .05       0 13761.1     .05       0 15620.6      .1       0
 17111.7      .1       0 19607.1     .05       0
Bank Sta=548.4,6859
XS Rating Curve= 0 ,0
Exp/Cntr=0.3,0.1

Type RM Length L Ch R = 1 ,254363  ,2607,2607,2607
BEGIN DESCRIPTION:
LOWER NUECES 51.0
END DESCRIPTION:
XS GIS Cut Line= 5
      2346678.17     13215105.13      2334834.09     13207068.07
      2335045.59     13202573.68      2332507.58     13197709.15
      2320082.94     13191311.78
#Sta/Elev= 30
-15949.7  138.11-12608.5  113.71-10979.2  127.24 -2573.1  133.45 -2423.3  132.02
 -2378.5  110.97 -2321.5  132.07 -2245.1   131.5 -1520.9  134.66  -886.5  132.97
  -237.7  134.07 1305.98   59.45    3032   65.05  3859.6   54.43  4622.6   51.69
  4720.7    57.9  4986.6   25.71  5149.3   26.44  5431.3   54.57    5440   53.13
  6040.3   48.85  6895.6   100.4  7461.6  123.898592.359  131.7310431.64  114.71
11191.34   135.4   12061  100.1712610.79  129.0513810.32  152.86 22324.9  180.97
#Mann= 19 ,-1 , 0
-15949.7     .05       0  -13876     .05       0-12750.5      .1       0
-12324.8     .05       0 -2245.1     .05       0 -1520.9     .05       0
  -886.5      .1       0  -237.7      .1       0  1318.1     .05       0
    3032     .16       0  3859.6     .12       0  4622.6     .05       0
    5440     .16       0  6895.6      .1       0  7461.6     .05       0
 12020.4      .1       0   13164      .1       0 14366.8      .1       0
 16015.4     .05       0
Bank Sta=4720.7,5431.3
XS Rating Curve= 0 ,0
Exp/Cntr=0.3,0.1

Type RM Length L Ch R = 1 ,251756  ,7621,7621,7621
BEGIN DESCRIPTION:
LOWER NUECES 52.0
END DESCRIPTION:
XS GIS Cut Line= 4
      2347418.38     13214470.59      2340808.99     13207596.83
      2333423.48     13194854.21      2324761.45     13190380.21
#Sta/Elev= 30
  -13805  141.18-13757.9  141.07-10548.4  122.81 -9868.7  107.18-8469.33  125.22
 -681.61  141.32-1.67968  135.73   986.1   88.71  1607.3   85.14  2442.1   60.02
 4297.68   57.79    4804    48.4  4965.9   26.01  5017.1   26.18  5069.9   54.55
5937.359   41.396207.311   56.197167.119      50  7613.7   60.35 9096.75   73.06
10656.48  123.9511826.46  125.9612526.46  139.6315616.42  132.1416026.41  142.23
16416.41  132.38 17106.4  146.6218176.39  141.14 19546.4  166.25 20208.3  170.69
#Mann= 16 ,-1 , 0
  -13805     .05       0-13757.9     .05       0 -9673.6     .05       0
 -4594.3     .05       0 -3486.4     .05       0 -3075.3      .1       0
 -2070.9     .05       0  2442.1     .05       0 8111.11     .05       0
  9390.6      .1       0 10225.5      .1       0 12111.2      .1       0
 12572.9     .05       0 16136.8      .1       0 17994.5     .05       0
 19546.4      .1       0
Bank Sta=2442.1,7613.7
XS Rating Curve= 0 ,0
Exp/Cntr=0.3,0.1

Type RM Length L Ch R = 1 ,244135  ,10235,10235,10235
BEGIN DESCRIPTION:
LOWER NUECES 53.0
END DESCRIPTION:
XS GIS Cut Line= 4
      2346394.23     13205999.07      2340426.76     13194227.62
      2337320.41     13192756.19      2325794.18      13190303.8
#Sta/Elev= 30
 -3109.8  126.39-1627.27  136.6872.43994  112.97792.3101  126.39 1292.22  108.31
 2082.08  102.72  3111.9   63.86 3761.79   77.86  4426.9   59.64  4901.4   52.91
  4998.4   24.94  5190.9   47.12 5841.41   55.36  7521.2   45.39  7902.1   58.02
  7968.9   64.44 8640.86  103.82 8920.81   91.93 9270.74  110.2510400.33  116.68
 12718.5  103.5413907.65  130.4615476.78  130.2916226.37  114.2118615.05  116.04
21153.65  150.1923072.59  140.6823892.14  155.79 25171.3  155.17 25309.3  156.76
#Mann= 16 ,-1 , 0
 -3109.8     .05       0  1715.6     .05       0  2069.1      .1       0
  2702.7     .16       0  3370.2      .1       0  4053.4     .05       0
 4211.81     .05       0  7968.9     .16       0  9134.1      .1       0
  9598.2     .16       0 10119.2     .05       0 14206.9     .05       0
 17896.2     .05       0 20419.3     .05       0 23089.9     .05       0
 25171.3      .1       0
Bank Sta=4426.9,7902.1
XS Rating Curve= 0 ,0
Exp/Cntr=0.3,0.1

Type RM Length L Ch R = 1 ,233900  ,7058,7058,7058
BEGIN DESCRIPTION:
Mapping XS 28f61c3d
END DESCRIPTION:
XS GIS Cut Line= 6
      2348659.38      13204487.7      2349026.25     13196992.92
      2347244.28     13195577.83      2338753.72     13192642.82
       2329005.3     13190022.27      2325755.79     13189865.04
#Sta/Elev= 30
   450.7  126.36 1691.97  130.36 2431.35  104.02  3986.4   87.82  4200.8   66.34
 4253.47   60.71  4408.2   43.04  4896.9   48.04  4996.7   23.58    5027   25.56
  5057.1   44.44  5137.1   46.57  6378.6   37.83  6488.8   52.87 7287.33   59.94
 7577.09   80.29  8705.3    73.8 9593.56   97.7814019.62   90.9614709.13  109.54
15548.54  105.6316567.81  119.1319815.41  100.7720564.97   125.721784.26  127.96
23063.51  108.8125701.96  112.9229708.99  150.16 32181.7  152.79 32561.3  157.24
#Mann= 16 ,-1 , 0
   450.7     .05       0  3986.4     .16       0  4200.8     .05       0
  6987.6     .16       0  6987.6      .1       0  9666.8     .05       0
 10948.4      .1       0 11986.7     .05       0 13096.7      .1       0
 13934.4      .1       0 14295.6     .05       0 16362.2      .1       0
 17508.1     .05       0 25078.5     .05       0 26466.4     .05       0
 32181.7      .1       0
Bank Sta=4253.47,7287.33
XS Rating Curve= 0 ,0
Exp/Cntr=0.3,0.1

Type RM Length L Ch R = 1 ,226842  ,4857,4857,4857
BEGIN DESCRIPTION:
LOWER NUECES 54.0
END DESCRIPTION:
XS GIS Cut Line= 6
      2356040.26     13208206.22      2354977.55      13202729.2
      2352606.92     13197987.94      2344677.55     13193410.16
      2331679.93     13188423.65      2323505.31     13189895.08
#Sta/Elev= 30
 -2846.6  124.65  722.47  121.15 1932.29    72.7 2772.11   81.35  4754.5   65.45
  4894.3   57.02  4961.4   26.25  5022.6   22.06  5095.5   46.21 6345.96   40.51
 7274.35   53.94 7374.17   59.41 8912.61   78.76  9562.3   69.6210032.07   83.78
11921.17    73.212640.83   98.1915999.44   86.5116679.17  109.6118458.23  105.27
19037.89   115.921496.45      9626763.36   94.6828582.29  103.9731220.54  144.68
32100.19  132.7334749.16  155.0636748.38  150.64 39210.6   180.9 39416.7  183.25
#Mann= 20 ,-1 , 0
 -2846.6     .05       0   825.1      .1       0  2512.7     .05       0
  4236.3      .1       0  4754.5     .07       0  4894.3     .05       0
 7274.35     .05       0  9601.4      .1       0 10787.2      .1       0
   11765     .05       0 14070.4     .05       0   14607      .1       0
 16427.8     .05       0 21623.7     .05       0 25807.2     .05       0
 28716.8     .05       0 35362.4     .12       0 36162.7     .05       0
 37176.6      .1       0 39210.6     .05       0
Bank Sta=4894.3,7374.17
XS Rating Curve= 0 ,0
Exp/Cntr=0.3,0.1

Type RM Length L Ch R = 1 ,221985  ,3456,3456,3456
BEGIN DESCRIPTION:
LOWER NUECES 54.5
END DESCRIPTION:
XS GIS Cut Line= 6
      2374760.08     13208860.14      2370264.06     13200603.81
      2354424.57     13197202.57      2345331.52      13192592.7
      2331679.93     13187687.94      2323670.73     13189485.92
#Sta/Elev= 30
-19148.6  130.59-10650.5  121.15-8466.96   99.92-7657.67  114.52-7098.16   94.21
-6698.51  113.62-4750.23  116.39-3730.37   86.84 1059.23    69.43089.061   82.76
  3568.5   80.76  3711.3   59.13    3750   55.41    4007   37.43  4914.4   45.07
  5023.3   20.61  5097.9    46.3  5381.4    33.9 5916.67   54.896358.801    73.1
11326.03   69.0111935.68    93.112865.15   72.2814924.21   74.63 17003.4  111.19
27189.42   95.6431377.84  157.4833187.57  136.56 37622.2   161.4 39366.5  177.09
#Mann= 19 ,-1 , 0
-19148.6     .05       0 -9360.1      .1       0 -6438.6      .1       0
 -5618.5     .05       0 -3545.2     .05       0 -1872.3      .1       0
   328.5      .1       0  1553.5      .1       0  3207.7      .1       0
  3711.3     .05       0 5916.67     .05       0  7042.3     .05       0
 10517.5      .1       0 11385.1     .05       0 13445.2     .16       0
 15161.9      .1       0 17211.7     .05       0 23985.5     .05       0
 37622.2      .1       0
Bank Sta=3750,5916.67
XS Rating Curve= 0 ,0
Exp/Cntr=0.3,0.1

Type RM Length L Ch R = 1 ,218529  ,12550,12550,12550
BEGIN DESCRIPTION:
LOWER NUECES 55.0
END DESCRIPTION:
XS GIS Cut Line= 4
      2376825.45     13209962.71      2371351.17     13200092.36
      2331723.79     13186623.54      2323377.75     13189189.05
#Sta/Elev= 30
-20867.1  125.01-12499.4  127.83-5760.85  107.25-3661.21  115.14-2511.43   84.82
 1147.85   86.28 1987.68   69.41 3687.35   78.16  4560.3   54.86  4565.6   53.65
  4924.7   46.75  4962.9   21.72    4994   19.87  5151.2   44.56  5742.1   34.74
    6500    54.6  6861.3   69.7611775.77   69.6512925.75   85.6715885.75   74.89
16835.75   83.0717475.75  106.1418395.75  109.8428475.75    95.631985.75  152.69
34413.38  141.06 39419.4  169.49 39780.9   180.2 40257.7  171.98 41004.9  170.22
#Mann= 19 ,-1 , 0
-20867.1     .05       0 -9830.6     .05       0 -7077.2      .1       0
 -5442.3     .05       0  -891.6     .05       0  1331.8     .05       0
  4565.6     .05       0    6500     .05       0  8810.6     .05       0
 12230.2     .05       0 14287.4      .1       0 15675.8      .1       0
 17564.2     .05       0 22008.9     .05       0 23228.9     .05       0
 31207.7     .05       0   37896      .1       0 39419.4      .1       0
 40257.7     .05       0
Bank Sta=4560.3,6500
XS Rating Curve= 0 ,0
Exp/Cntr=0.3,0.1

Type RM Length L Ch R = 1 ,205979  ,12337,12337,12337
BEGIN DESCRIPTION:
LOWER NUECES 56.0
END DESCRIPTION:
XS GIS Cut Line= 5
      2384195.58      13197611.4      2366610.99     13189541.08
      2350927.69     13187137.76      2331261.52     13181034.36
       2327053.6     13179131.51
#Sta/Elev= 30
-24145.8  118.03-17105.2  115.91-6185.77  110.44-1996.46   70.89802.9902   65.03
1762.801   42.072692.619   48.863072.539   42.293112.539   30.75 3232.51   44.48
 4622.24   43.72  4927.8   38.14  4965.5   19.85  5018.6   16.42  5109.9   44.78
  5635.9    36.1  5692.8   48.25  5824.6   58.57 7101.76   51.949651.059   72.66
16668.32   59.2720017.01   69.2822745.94   93.9626154.61   94.7926504.47   82.17
29123.45  102.29 31562.5  140.3834071.52  137.3335361.01  160.38 36278.3  154.34
#Mann= 17 ,-1 , 0
-24145.8     .05       0-17105.2     .05       0   -9341     .05       0
 -5147.5     .05       0 -2185.2      .1       0  -709.6     .05       0
  1062.5     .05       0  5692.8     .05       0  7592.7     .05       0
 14432.5     .05       0 23825.7      .1       0 24951.4     .05       0
 26737.1     .05       0 28435.1     .05       0 31875.5      .1       0
 34142.3     .05       0 35509.6      .1       0
Bank Sta=2692.619,5692.8
XS Rating Curve= 0 ,0
Exp/Cntr=0.3,0.1

Type RM Length L Ch R = 1 ,193642  ,9153,9153,9153
BEGIN DESCRIPTION:
LOWER NUECES 57.0
END DESCRIPTION:
XS GIS Cut Line= 4
      2375696.49     13184486.68      2360545.69     13177790.08
        2341352.      13177240.5       2329312.1     13178955.15
#Sta/Elev= 30
-18206.6  112.18-10576.4  111.27-8527.03   98.77-7457.35  107.31-7067.46  105.99
 -4548.2   45.79 2009.51   46.63 3338.99   34.94 3708.84   43.53  4898.8   41.46
  4968.8    15.3  5008.6   14.49  5108.9    35.2 5428.17   41.12 6757.65   32.75
 6937.58   42.247507.359   42.878287.051   31.88 8616.93   47.06 9656.52   36.19
10716.11   70.6713065.19   70.2314194.75   86.1316523.84    94.720521.12    85.1
22129.86   95.49 22969.2  112.83 27155.1  121.31 28936.8  136.77 29721.1  143.93
#Mann= 18 ,-1 , 0
-18206.6     .05       0 -8022.8     .05       0 -7191.8      .1       0
 -6290.6      .1       0 -5300.2     .16       0 -4407.3     .05       0
    33.1     .16       0  1797.5     .05       0  8900.4     .05       0
 11575.1     .05       0 16297.9     .05       0 19006.8     .16       0
 19898.5      .1       0 20655.6     .05       0 25476.1     .05       0
   26316      .1       0 27155.1     .05       0 28936.8      .1       0
Bank Sta=2009.51,8616.93
XS Rating Curve= 0 ,0
Exp/Cntr=0.3,0.1

Type RM Length L Ch R = 1 ,184489  ,4540,4540,4540
BEGIN DESCRIPTION:
LOWER NUECES 58.0
END DESCRIPTION:
XS GIS Cut Line= 4
      2376219.35     13184072.46      2348461.43     13171856.55
      2336143.67     13177111.94      2329210.95      13178537.7
#Sta/Elev= 30
-21678.3  111.63-12894.8  109.36-11684.9   93.72  -11015  106.86-9275.18   56.53
 -8005.3   44.56 -2815.8   47.26 -1675.9   31.18263.9102   46.181643.779   47.04
 1883.76   32.75    2924   41.94  4828.9   35.86  4911.3   33.57  4986.5   11.39
  5038.9   12.21  5108.9   38.78    5750   42.39 6483.33   66.31 7283.25   71.19
12420.84    57.613250.31   67.9713809.95   90.54 20465.7   91.8721674.92  117.53
 22524.5  119.2525263.43  105.53 26986.3  130.82 27603.4  135.84 29118.6  145.92
#Mann= 19 ,-1 , 0
-21678.3     .05       0-10935.7      .1       0 -7529.1     .05       0
 -4163.3      .1       0 -1602.7      .1       0  -436.9      .1       0
   715.8     .16       0  1488.4      .1       0    2073     .16       0
    2924     .05       0    5750     .16       0  7819.4     .05       0
 12697.1     .05       0 16564.6     .05       0 20225.1      .1       0
 20748.2     .05       0 25988.9      .1       0 26986.3     .05       0
 27603.4      .1       0
Bank Sta=2924,5750
XS Rating Curve= 0 ,0
Exp/Cntr=0.3,0.1

Type RM Length L Ch R = 1 ,179949  ,9606,9606,9606
BEGIN DESCRIPTION:
LOWER NUECES 59.0
END DESCRIPTION:
XS GIS Cut Line= 3
      2377138.51     13176992.73      2348790.61     13168315.98
      2333533.62     13167150.61
#Sta/Elev= 30
-20600.5  105.07-12175.1  108.37-9775.38   53.22 -6773.4   42.34 -6175.9   43.89
 -5799.8   20.89 -4954.6   57.24 -4643.7   24.32 -4295.1   44.09 -2836.7   35.96
  -874.2   41.67   549.8   31.82   818.2   42.28   880.9   23.13  1090.1    50.7
  3295.9   33.11  4254.4   37.11  4907.2   37.19  4924.2    29.3    4957   11.35
  5060.5   29.53  5074.6   36.77  5823.8   29.52 8171.57   61.1911709.83   56.33
 14878.5   87.3716397.91   62.0417327.55  115.3519726.61   99.31   24347  147.86
#Mann= 20 ,-1 , 0
-20600.5     .05       0-12849.8     .05       0-10730.7     .05       0
 -9819.8      .1       0 -8400.8     .05       0 -6773.4      .1       0
 -2836.7      .1       0  -874.2     .16       0   549.8     .16       0
  3295.9     .16       0  4254.4     .16       0  4924.2     .05       0
  5060.5     .16       0  5823.8     .16       0  8095.9     .05       0
  9801.2     .05       0 13649.8     .16       0 16953.5     .05       0
 18203.2      .1       0 19922.9     .05       0
#XS Ineff= 2 , 0
        -4959.79   57.42
Permanent Ineff=
       F       F
Bank Sta=4907.2,5074.6
XS Rating Curve= 0 ,0
Exp/Cntr=0.3,0.1

Type RM Length L Ch R = 1 ,170343  ,19624,19624,19624
BEGIN DESCRIPTION:
LOWER NUECES 61.0
END DESCRIPTION:
XS GIS Cut Line= 6
      2375217.89     13175577.16      2370306.31     13170873.08
      2361841.75     13168072.79      2351103.15     13162396.39
      2341398.15     13158426.64      2338971.65     13157721.05
#Sta/Elev= 30
-19953.6  105.57-17013.5  106.53-12593.3  107.18-10564.3   40.75 -6016.6   42.71
-5566.82   24.02-4857.16    46.3-3087.81      45-2418.02   16.59 -2158.1   39.26
-1038.44   42.31  2020.6    47.12520.449   21.28  4929.6   31.34  5033.8   10.91
    5479   32.83    5501   32.77  5885.9   27.58    6018   79.44    6062   51.43
7069.039   41.62 7159.01   -1.27 7248.98   23.517588.869   26.037638.859    5.59
 7688.84   35.19 10387.8   31.7613356.64  109.03 19934.1  116.12 20922.1  112.98
#Mann= 20 ,-1 , 0
-19953.6     .05       0-17013.5     .05       0  -12195      .1       0
-10231.7     .05       0 -6589.7      .1       0 -5422.9     .12       0
 -4789.7     .05       0 -1131.7     .05       0   617.2     .05       0
  2540.5     .16       0  5033.8     .05       0    5501     .05       0
  7154.9     .07       0  7160.9     .05       0   10191     .12       0
 11975.9      .1       0   12949      .1       0 14753.7     .05       0
 16092.9     .05       0 19934.1     .05       0
#XS Ineff= 2 , 0
                         6005.36           79.72
Permanent Ineff=
       F       F
Bank Sta=4929.6,5479
XS Rating Curve= 0 ,0
Exp/Cntr=0.3,0.1

Type RM Length L Ch R = 1 ,150719  ,7252,7252,7252
BEGIN DESCRIPTION:
LOWER NUECES 62.0
END DESCRIPTION:
XS GIS Cut Line= 5
      2375688.67     13175162.67       2369918.8     13167830.76
      2361090.49     13163732.18      2355899.88     13159818.24
      2341833.41      13152806.6
#Sta/Elev= 30
-11362.3  105.38-4664.03  102.55-1304.56   29.85 4176.86    30.8  4927.2    28.9
  5018.6    5.33  5470.4   29.948467.971   29.368537.881   30.5811617.69   36.66
12556.41   18.1812955.86   36.7514124.26   18.1814204.15   34.1515083.98   35.07
15123.97   13.4115883.82   13.3916063.79   40.57 17456.3   40.57 17536.6   73.91
 17805.2   80.4118099.39   31.0719279.16   34.2419339.14   12.6619889.04   12.66
19999.02   30.7722258.73   21.4423328.73   44.2124688.71  106.95   29919  107.78
#Mann= 18 ,-1 , 0
-11362.3     .05       0 -4925.1     .05       0   -4014     .05       0
 -2769.8     .05       0  -695.9     .05       0   663.2      .1       0
    2884      .1       0  4927.2     .05       08467.971     .16       0
  9023.3      .1       0  9801.5      .1       0 10714.8     .16       0
 13488.1     .05       0 14395.4      .1       0 15110.2     .05       0
 17456.3     .05       0 21773.8      .1       0 25267.8     .05       0
#XS Ineff= 2 , 0
                        17801.61           80.61
Permanent Ineff=
       F       F
Bank Sta=4176.86,8537.881
XS Rating Curve= 0 ,0
Exp/Cntr=0.3,0.1

Type RM Length L Ch R = 1 ,143467  ,6307,6307,6307
BEGIN DESCRIPTION:
LOWER NUECES 63.0
END DESCRIPTION:
XS GIS Cut Line= 4
      2377823.07     13175433.29      2374087.89     13167065.84
      2365131.56     13161042.56      2343172.03     13148923.76
#Sta/Elev= 30
-11725.9  104.77-5893.27  106.55-5033.89   96.53-3305.15   17.82-2465.75      33
-1996.04   16.33222.6201   35.04292.5801   19.41  4909.2   27.79  4966.8    4.58
    5198   26.08 17835.2    25.8 17932.1   44.97 18025.4   35.21   18085   61.12
 18166.4   35.46 18247.7   56.45 18334.8   30.08 18513.6   40.98 18747.4    21.1
 23971.7   18.0124171.62   37.6824881.34   18.9624931.32   33.8926300.79   41.81
 27040.5   90.5227750.22  105.5628769.82   85.8629509.53  105.95 33312.3   105.5
#Mann= 19 ,-1 , 0
-11725.9     .05       0 -5524.5      .1       0   -4769     .05       0
 -2187.6     .16       0   -1006     .05       0   909.8     .12       0
  3872.2     .05       0    5198     .16       0  6258.9     .05       0
  7030.6     .16       0    8574     .16       0 10889.6      .1       0
   11573      .1       0 13085.4     .05       0 20943.7      .1       0
   21728     .05       0 22797.8     .05       0 25900.5      .1       0
 29147.9     .05       0
Bank Sta=4909.2,5198
XS Rating Curve= 0 ,0
Exp/Cntr=0.3,0.1

Type RM Length L Ch R = 1 ,137160  ,5964,5964,5964
BEGIN DESCRIPTION:
LOWER NUECES 64.0
END DESCRIPTION:
XS GIS Cut Line= 6
      2380064.11      13175183.5      2374627.25     13163914.59
      2363895.59     13156200.92      2360613.56     13152582.41
      2358373.31     13139765.79      2358552.25     13136226.32
#Sta/Elev= 30
-15245.1   103.3-14008.2  101.37 -8320.5   95.21 -5506.6   32.97 -5422.6   19.33
 -4989.6   20.66 -4907.7   36.64 -4834.2   37.06-786.669    29.1422.9697   41.97
   662.8   33.23    1103   22.81  3325.1   25.58  4901.9   26.19  5002.3    4.21
    5111   23.39  5491.1   19.39  5541.4   27.01  9485.5   25.34 11560.3   21.94
 12581.6   21.66 13535.8   18.76 15262.3   52.55 18155.5   56.23 19008.2   71.69
 19930.6   64.63 21999.4   72.49 22430.5   72.66 23924.3   73.25 31923.2    91.9
#Mann= 17 ,-1 , 0
-15245.1     .05       0-14008.2     .05       0 -4546.4     .05       0
   662.8     .16       0    1103     .12       0  3325.1     .12       0
  4901.9     .05       0  7030.4     .16       0  8868.9      .1       0
  9485.5      .1       0 11560.3     .16       0 12581.6     .16       0
 15262.3     .05       0 19930.6     .05       0 21999.4      .1       0
 22430.5     .05       0 23924.3     .05       0
#XS Ineff= 2 , 0
                         7939.79            28.2
Permanent Ineff=
       F       F
Bank Sta=4901.9,5541.4
XS Rating Curve= 0 ,0
Exp/Cntr=0.3,0.1

Type RM Length L Ch R = 1 ,131196  ,5875,5875,5875
BEGIN DESCRIPTION:
LOWER NUECES 65.0
END DESCRIPTION:
XS GIS Cut Line= 4
      2380378.86     13174716.19      2375545.19     13161514.39
      2364616.36     13148335.51      2363146.35     13139733.29
#Sta/Elev= 30
-15613.8  102.72-11304.7  104.96 -6967.4   83.52 -6173.1    35.1 -5465.8   19.32
 -5221.8   23.88 -3696.4   35.04   573.8   22.82   813.6   13.65   934.7   22.55
  1701.8      14    2546   21.81  4904.1   23.53  4953.3    4.04  5060.4    4.55
  5117.7   23.67  5471.4   23.54  6677.8   21.73  9321.5    18.4 10862.8   20.31
 11836.3   21.51 13576.2   49.81 14918.4   71.66 16178.9   71.92 16856.8   71.82
 17892.5   70.49 19389.7   74.56 21518.4   86.12 22403.6   89.08 24292.8   94.32
#Mann= 19 ,-1 , 0
-15613.8     .05       0-11304.7     .05       0 -5221.8     .05       0
   573.8     .12       0    2546     .05       0  5471.4     .05       0
  5471.4     .16       0  6677.8     .05       0  9321.5     .05       0
 10862.8     .05       0 11836.3     .05       0 13576.2     .05       0
 14918.4      .1       0 16178.9     .05       0 16856.8     .05       0
 17892.5     .05       0 19389.7     .05       0 21518.4     .05       0
 22403.6     .05       0
#XS Ineff= 2 , 0
        -3453.98   35.18
Permanent Ineff=
       F       F
Bank Sta=4904.1,5117.7
XS Rating Curve= 0 ,0
Exp/Cntr=0.3,0.1

Type RM Length L Ch R = 1 ,125321  ,13753,13753,13753
BEGIN DESCRIPTION:
LOWER NUECES 66.0
END DESCRIPTION:
XS GIS Cut Line= 4
      2380850.39     13174145.44      2377896.66     13159962.84
      2375529.79     13153232.42      2375299.11     13136561.49
#Sta/Elev= 30
-14674.7   103.6 -8492.2  100.26 -8068.7   85.18 -7769.5   88.04 -7214.3   96.88
 -6698.6   84.46   -6328   57.41 -5697.9   40.32 -3318.3   34.16 -2243.1   31.04
 -1540.5   32.56 -1125.6   30.53   422.2   24.06   465.2   21.45   963.4   12.34
  4874.9   22.58  4927.9   16.42  4945.9    3.92  5055.1    4.42    5101   23.14
  5281.5    23.8  5338.1   20.52  7652.3    20.6  7752.3   10.36 10842.1   17.37
 11262.7    41.3 12518.5    48.7 20923.6   92.31 23602.2   91.74 23619.2   91.64
#Mann= 15 ,-1 , 0
-14674.7     .05       0 -8492.2      .1       0 -7769.5      .1       0
 -7214.3     .16       0   -6328     .16       0 -5697.9     .05       0
 -3318.3     .05       0 -2243.1     .16       0 -1540.5     .16       0
 -1125.6     .05       0   465.2     .05       0  5338.1     .05       0
 10842.1      .1       0 12518.5     .05       0 23602.2     .05       0
Bank Sta=422.2,5281.5
XS Rating Curve= 0 ,0
Exp/Cntr=0.3,0.1

Type RM Length L Ch R = 1 ,111568  ,4104,4104,4104
BEGIN DESCRIPTION:
LOWER NUECES 67.0
END DESCRIPTION:
XS GIS Cut Line= 3
      2386961.14     13170736.66      2383923.43     13163273.26
      2379672.76     13137051.57
#Sta/Elev= 30
-13826.3   97.74 -8060.2   97.25 -5654.4   98.64 -5217.2   97.79 -4566.5   61.79
 -4191.7   74.42 -3829.3   38.11-3561.22   22.07  1440.9   15.81  1592.9    6.61
  1653.7   16.87  4885.3   17.78  4953.2    4.29  5049.9    4.69  5087.9   19.21
  5671.4    13.5    6334   22.33  6708.8   29.42  6789.8   10.87  6862.8    9.34
  6931.7   31.16  7263.4   22.57  9413.7   37.16 10082.3    81.9   11068    86.7
 11959.8   82.95 12406.1   79.83   13275   88.04 14889.2   92.22 20795.6   94.91
#Mann= 12 ,-1 , 0
-13826.3     .05       0 -8060.2     .05       0 -5654.4     .16       0
 -5217.2      .1       0-3561.22     .05       0    6334      .1       0
  7263.4     .05       0   11068     .16       0 11959.8     .16       0
 12406.1     .16       0   13275     .05       0 14889.2     .05       0
Bank Sta=-3561.22,6334
XS Rating Curve= 0 ,0
Exp/Cntr=0.3,0.1

Type RM Length L Ch R = 1 ,107464  ,8712,8712,8712
BEGIN DESCRIPTION:
LOWER NUECES 68.0
END DESCRIPTION:
XS GIS Cut Line= 4
      2390904.29     13169232.92      2390651.52     13160131.33
      2382555.45     13144769.78       2381579.5     13136383.92
#Sta/Elev= 30
-15018.9   96.92 -8317.9   70.07 -7625.1   68.97 -5700.8   63.87 -5277.2   35.52
   -5120   37.04 -4842.2   44.22 -4370.5   28.21 -2788.2   19.16 -2370.6    8.15
 -1287.4    7.85 -1221.3   14.56   473.7   15.55     591    8.47   726.6   16.04
  4920.4   17.85  4958.8    4.35    5019    3.75  5145.8   17.92  6912.5   22.03
  6972.9   25.71  7344.8   49.85  7578.4   68.13  8007.6   83.02    8634   86.65
  9508.3   87.53 10002.1   79.05 13318.9   94.97 16215.3   96.66 19893.1   94.98
#Mann= 13 ,-1 , 0
-15018.9     .05       0 -8317.9     .05       0 -7625.1     .05       0
   -5120      .1       0 -4370.5     .16       0 -2788.2     .05       0
  6972.9     .12       0  7344.8      .1       0    8634     .05       0
  9508.3      .1       0 10002.1     .05       0 13318.9     .05       0
 16215.3     .05       0
Bank Sta=-2788.2,6912.5
XS Rating Curve= 0 ,0
Exp/Cntr=0.3,0.1

Type RM Length L Ch R = 1 ,98752   ,9406,9406,9406
BEGIN DESCRIPTION:
LOWER NUECES 69.0
END DESCRIPTION:
XS GIS Cut Line= 4
      2392881.02     13169051.03      2392404.25     13159828.68
      2391227.28     13149964.72      2388751.34     13136204.69
#Sta/Elev= 30
-12999.4   94.19-11724.5   84.45 -7606.5   81.75 -5389.3   68.97 -3663.9   51.25
-1773.91   18.52  -600.6    8.94  3790.3   15.27  3820.5    5.94  3870.9   14.12
  4942.5   15.29  4968.4    3.67    5019    4.88  5049.2   16.52  8055.1   13.84
  8097.5      19    8128    9.92  8231.2    8.71  8321.1   33.46    8382    9.32
  8756.4   11.87  9773.8   12.46 11221.2   13.31 11591.4   34.81 12019.5   49.27
 12601.2   35.29 13280.1   60.09 15555.4   85.23 17953.4      92 20150.2    89.6
#Mann= 13 ,-1 , 0
-12999.4     .05       0-11724.5     .05       0 -7606.5      .1       0
 -5389.3     .05       0 -3663.9      .1       0-1773.91     .05       0
  8055.1     .12       0  8756.4     .05       0  9773.8     .07       0
 11591.4      .1       0 12601.2      .1       0 13280.1     .05       0
 17953.4     .05       0
#XS Ineff= 2 , 0
                         8333.33           33.12
Permanent Ineff=
       F       F
Bank Sta=-1773.91,8097.5
XS Rating Curve= 0 ,0
Exp/Cntr=0.3,0.1

Type RM Length L Ch R = 1 ,89346   ,12043,12043,12043
BEGIN DESCRIPTION:
LOWER NUECES 70.0
END DESCRIPTION:
XS GIS Cut Line= 3
      2393838.56     13166368.77      2396868.84     13157229.04
      2392250.34     13135631.22
#Sta/Elev= 30
-12847.6   95.77-10716.6   86.64 -9984.3    83.5 -9054.8   79.52 -8180.8   71.09
   -6851    51.9 -5331.3   51.48 -4512.9   51.25 -3595.6      51 -3141.2   17.63
-3114.39    16.6  4913.4   12.84  5005.1    3.58  5082.9   12.85  5506.5    7.84
  5547.4   14.86  6278.9     7.6  8913.1   16.69  8957.5   17.37  9954.8    9.79
 10159.3   18.01   10190    11.3 11069.5   21.47 12195.1   18.52 12920.4    23.5
 13306.4    43.3 13713.6   48.93 16170.5   71.65 17587.2   87.05 18867.5   91.11
#Mann= 13 ,-1 , 0
-12847.6     .05       0-10716.6     .16       0 -9984.3      .1       0
 -9054.8     .05       0 -8180.8      .1       0 -5331.3     .16       0
 -4512.9      .1       0 -3141.2     .05       0  8957.5      .1       0
 12195.1     .05       0 13713.6     .05       0 16170.5     .05       0
 17587.2     .05       0
Bank Sta=-3114.39,8913.1
XS Rating Curve= 0 ,0
Exp/Cntr=0.3,0.1

Type RM Length L Ch R = 1 ,77303   ,7226,7226,7226
BEGIN DESCRIPTION:
LOWER NUECES 71.0
END DESCRIPTION:
XS GIS Cut Line= 6
      2395041.43     13167169.44      2396862.86     13163913.79
      2399116.85     13160597.62      2402172.34      13149790.1
      2396988.13     13139261.78      2395542.58      13135083.6
#Sta/Elev= 30
  -22398   70.89-22052.1   86.09-21392.1   91.28  -20405   67.83-19916.3   81.96
-18559.4   88.41-17849.5   55.63-17109.6   38.21-16429.6   56.32-15819.7   49.64
-15239.7   57.22-14619.8   42.12-13960.3   44.71-13470.7   14.15-13330.8   12.53
-9363.96     4.3-7685.28   14.95-5257.17   14.06-2808.85   23.98-1685.27   12.72
  4810.5   11.31  4967.5    3.46  5147.5   13.19  5242.9   20.12 5447.93   16.88
 6077.68   55.029264.939   62.7810113.28   57.63 12508.8   88.74   12730   89.12
#Mann= 18 ,-1 , 0
  -22398      .1       0  -19220      .1       0-16540.9      .1       0
-14964.9      .1       0-13441.9     .12       0-11843.7     .05       0
 -8127.2      .1       0 -5213.6     .12       0 -4329.1     .16       0
   -3200     .07       0 -2404.6      .1       0 -1683.2     .05       0
  5377.7     .05       0  6205.1     .05       0    8626     .08       0
  9724.4     .05       0   11099     .05       0 12508.8     .05       0
Bank Sta=-1685.27,5147.5
XS Rating Curve= 0 ,0
Exp/Cntr=0.3,0.1

Type RM Length L Ch R = 1 ,70077   ,8767,8767,8767
BEGIN DESCRIPTION:
LOWER NUECES 72.0
END DESCRIPTION:
XS GIS Cut Line= 6
      2395031.13     13168074.87      2397816.08     13164398.44
      2400168.01     13160502.91      2404509.09     13149182.99
      2405273.72      13136868.9      2404112.29     13130190.33
#Sta/Elev= 30
-25530.9   71.02-25392.5   62.02-25099.1   76.31-24699.9   60.03-23592.9   76.99
-22900.2   49.88-22221.9   78.96-21992.1   75.76-21780.8   63.44-21469.9   79.47
-20421.3   80.09-19828.3   58.55-18971.9    50.9  -18463   27.45-17375.2   48.64
  -16547   50.62-16077.5   46.99-15647.7    16.7-12339.3    4.151235.119    4.44
    1855   13.01  4959.1    3.36  5089.6   10.576314.131   13.17  7634.5   63.05
  8532.2   78.87 10927.8   84.88 12037.4   84.13   14660   80.85 14872.1   80.45
#Mann= 15 ,-1 , 0
-25530.9      .1       0-24699.9      .1       0-22900.2      .1       0
-21992.1     .05       0-21469.9      .1       0-19828.3     .16       0
-18986.7      .1       0-17092.3      .1       0-14234.2     .05       0
  5089.6     .07       0    6579     .05       0  8532.2      .1       0
 10927.8     .05       0 12037.4     .05       0   14660     .05       0
Bank Sta=1855,6314.131
XS Rating Curve= 0 ,0
Exp/Cntr=0.3,0.1

Type RM Length L Ch R = 1 ,61310   ,9704,9704,9704
BEGIN DESCRIPTION:
LOWER NUECES 73.0
END DESCRIPTION:
XS GIS Cut Line= 4
      2402028.02     13172605.25      2402189.25      13160729.4
      2412368.47     13138274.59      2411383.27     13127532.22
#Sta/Elev= 30
-29942.8   96.63-25737.8   98.46-24749.6   98.87-24663.9  111.25-24613.9   97.91
-22066.5   91.68-19709.9   66.51-18431.6   49.13-17853.1   47.63-17123.3   12.91
-16973.3   11.37-3436.05    2.83  4999.8    3.69  5051.5   12.93  5092.2   33.26
  5126.2   65.25  5257.4   58.26  5334.1    41.7  5633.1   75.18  5839.4   80.98
    7830   80.64  9626.4   81.93 10321.8   79.31 10392.1   93.42   10603   94.53
 10705.6   81.26 12983.4    76.9 13213.9   68.77 14874.9   75.62 17375.9    73.9
#Mann= 12 ,-1 , 0
-29942.8     .05       0-25737.8     .08       0-24749.6     .05       0
-22066.5      .1       0-19709.9      .1       0-18431.6      .1       0
-16973.3     .05       0  4999.8     .07       0    7830     .05       0
  9626.4     .15       0 12983.4     .05       0 14874.9     .05       0
Bank Sta=-17123.3,5051.5
XS Rating Curve= 0 ,0
Exp/Cntr=0.3,0.1

Type RM Length L Ch R = 1 ,51606   ,763,763,763
BEGIN DESCRIPTION:
LOWER NUECES 74.0
END DESCRIPTION:
XS GIS Cut Line= 6
      2402568.68     13170082.54      2402507.44     13166566.13
      2408390.83     13154410.86      2412915.65     13143745.09
      2413279.91     13137526.07      2412196.86     13127181.04
#Sta/Elev= 30
-18570.1   96.62-15615.3   95.59-11975.1   82.08-10516.1   94.18-9576.76   58.24
-9067.11   71.19 -7168.4      18-5769.43   10.09    3092   11.13  3138.4   11.22
  4907.9    -.07 9003.35   11.8511265.66   20.1212751.33   53.4212881.08   31.56
13988.91   55.8114847.23   47.78 15464.3   75.34 15929.3   72.75 16543.6      63
 16887.7   83.28 17088.8   68.65 17259.7   97.32 17390.5   75.92 18642.4   90.37
 20006.7    94.1 21060.4   75.27 22507.4   75.69 23580.5   76.53 26686.8    73.6
#Mann= 19 ,-1 , 0
-18570.1     .05       0-15615.3     .05       0-12804.2      .1       0
   -7189     .05       0 -3824.8      .1       0 -2814.4     .07       0
    50.7     .07       0  1404.1     .07       0    3092     .05       0
  8753.1     .07       0  8893.7     .05       0  9795.6     .15       0
 11605.5     .15       0   12427     .15       0 15929.3     .08       0
 18642.4     .05       0 21060.4      .1       0 22507.4     .05       0
 23580.5     .05       0
Bank Sta=3138.4,9003.35
XS Rating Curve= 0 ,0
Exp/Cntr=0.3,0.1

Type RM Length L Ch R = 1 ,50843   ,2480,2480,2480
BEGIN DESCRIPTION:
LOWER NUECES 75.0
END DESCRIPTION:
XS GIS Cut Line= 6
      2403137.78     13167684.72      2409123.55     13156423.86
      2413415.51     13143546.55      2414003.39     13138308.48
      2413096.19     13134375.39      2412349.55      13127165.4
#Sta/Elev= 30
-15963.7   96.38-15001.2   95.65  -13591   95.66-12232.7   94.85 -9753.8   91.26
   -8087   39.48 -7425.5   33.88 -4246.4   11.29 -3265.2    9.93 -1046.8   11.45
    2904    8.25  2936.2    9.09  4875.5    -.13    6637    11.3  6640.9   11.31
  9181.4   14.73 11701.1    8.46 13079.4   13.55 14429.3    20.1   15646   66.13
 16181.2   55.21 16490.9   82.34   16768   48.94   16987   59.41 17168.4  104.62
 17465.8   64.82 19328.5   90.82 22633.9   72.54 23888.5    75.6 26932.6   73.16
#Mann= 18 ,-1 , 0
-15963.7     .05       0-15001.2     .05       0  -13591     .05       0
-12232.7      .1       0   -8087     .16       0 -7425.5      .1       0
 -4246.4     .05       0 -3265.2     .07       0 -1046.8      .1       0
    2904     .05       0  6640.9     .07       0  6640.9      .1       0
  9181.4      .1       0 11701.1      .1       0 13079.4     .16       0
 19328.5     .05       0 22633.9     .05       0 23888.5     .05       0
#XS Ineff= 2 , 0
                        10798.61           22.52
Permanent Ineff=
       F       F
Bank Sta=2936.2,6637
XS Rating Curve= 0 ,0
Exp/Cntr=0.3,0.1
