--- PAISANO CREEK.prj (project) ---

Proj Title=PAISANO CREEK Base Level Engineering
Current Plan=p01
Default Exp/Contr=0.3,0.1
English Units
Geom File=g01
Flow File=f01
Plan File=p01
Y Axis Title=Elevation
X Axis Title(PF)=Main Channel Distance
X Axis Title(XS)=Station
BEGIN DESCRIPTION:
PAISANO CREEK
END DESCRIPTION:
DSS Export Rating Curves= 0
DSS Export Rating Curve Sorted= 0
DSS Export Volume Flow Curves= 0
DXF OffsetX= 0
DXF OffsetY= 0
DXF ScaleX= 1
DXF ScaleY= 10

--- PAISANO CREEK.p01 (plan) ---

Plan Title=Multiple Run
Short Identifier=Multiple
Geom File=g01
Flow File=f01
Subcritical Flow
K Sum by GR= 0
Std Step Tol= 0.01
Critical Tol= 0.01
Num of Std Step Trials= 20
Max Error Tol= 0.3
Flow Tol Ratio= 0.001
Split Flow NTrial= 30
Split Flow Tol= 0.02
Split Flow Ratio= 0.02
Log Output Level= 0
Friction Slope Method= 1
Unsteady Friction Slope Method= 2
Unsteady Bridges Friction Slope Method= 1
Parabolic Critical Depth
Global Vel Dist=  1 , 1 , 1
Global Log Level= 0
CheckData=True
Encroach Param= -1, 0, 0, 0
BEGIN DESCRIPTION:
Multiple Run
END DESCRIPTION:

--- PAISANO CREEK.f01 (steady flow) ---

Flow Title=Multiple
Program Version=4.10
Number of Profiles= 7
Profile Names=10-year,25-year,50-year,1pct_min,100-year,1pct_plu,500-year
River Rch & RM=PAISANO CREEK,Reach-1         ,25638
     273     386     482     444     600     812     945
River Rch & RM=PAISANO CREEK,Reach-1         ,21482
     479     691     875     813    1100    1488    1765
River Rch & RM=PAISANO CREEK,Reach-1         ,13336
    1217    1798    2309    2169    2933    3967    4796
River Rch & RM=PAISANO CREEK,Reach-1         ,5250
    1341    1982    2545    2388    3239    4367    5264
Boundary for River Rch & Prof#=PAISANO CREEK,Reach-1         , 1
Up Type= 0
Dn Type= 3
Dn Slope=0.005
Boundary for River Rch & Prof#=PAISANO CREEK,Reach-1         , 2
Up Type= 0
Dn Type= 3
Dn Slope=0.005
Boundary for River Rch & Prof#=PAISANO CREEK,Reach-1         , 3
Up Type= 0
Dn Type= 3
Dn Slope=0.005
Boundary for River Rch & Prof#=PAISANO CREEK,Reach-1         , 4
Up Type= 0
Dn Type= 3
Dn Slope=0.005
Boundary for River Rch & Prof#=PAISANO CREEK,Reach-1         , 5
Up Type= 0
Dn Type= 3
Dn Slope=0.005
Boundary for River Rch & Prof#=PAISANO CREEK,Reach-1         , 6
Up Type= 0
Dn Type= 3
Dn Slope=0.005
Boundary for River Rch & Prof#=PAISANO CREEK,Reach-1         , 7
Up Type= 0
Dn Type= 3
Dn Slope=0.005
DSS Import GetInterval= 0
DSS Import GetPeak= 0
DSS Import FillOption= 0

--- PAISANO CREEK.g01 (geometry) ---

Geom Title=Existing Conditions
Program Version=4.10

River Reach=PAISANO CREEK   ,Reach-1
Reach XY= 30
      2284032.72     13267651.85      2284561.65     13269195.14
      2285056.06     13269977.21      2286015.36     13270375.68
      2286547.04      13269974.2      2288059.31     13270826.55
      2288988.16     13270211.28      2289512.59      13269073.3
      2289930.67     13268742.35      2290181.71     13268002.07
      2290603.96     13267597.02      2291346.53     13267593.97
      2291873.14     13267217.33      2292740.19     13267412.27
      2293822.58     13268604.27      2294375.61     13269568.08
      2294420.85      13269920.3      2295738.69     13270738.04
      2295905.06     13271182.31      2296643.46     13271605.06
       2298112.7     13271448.07      2298316.63     13271546.82
      2298526.48     13271986.34      2298463.25     13272519.56
      2299187.91     13272936.87      2299066.38     13273787.56
      2299266.03      13274497.2      2299077.23     13275167.77
      2298686.98     13275590.23      2299044.62     13275645.79

Type RM Length L Ch R = 1 ,25638   ,206,206,206
BEGIN DESCRIPTION:
PAISANO CREEK 42.0
END DESCRIPTION:
XS GIS Cut Line= 3
      2283937.75     13268146.83      2284237.72     13267896.85
      2284537.69     13267696.87
#Sta/Elev= 30
  4641.4   230.1  4669.4  229.38  4705.8  227.16  4755.3  221.73  4797.6  220.44
  4804.7  219.59  4839.9  218.36  4847.7  217.64  4889.3  216.76  4897.1  216.06
    4918  216.19    4932  215.01  4953.8  217.41  4960.9  217.01  4975.3  216.03
  4981.8  216.42  5003.9  216.16  5010.4  216.62  5096.5  219.02  5111.5  220.12
  5153.6  221.69  5189.6  224.49  5204.6  224.88  5255.7  228.36  5276.8  229.04
  5297.8  231.14  5333.8  233.03  5363.9   235.6  5378.9  235.96  5392.4  237.27
#Mann= 3 , 0 , 0
  4641.4     .16       0  4960.9     .07       0  5010.4     .16       0
Bank Sta=4960.9,5010.4
XS Rating Curve= 0 ,0
Exp/Cntr=0.3,0.1

Type RM Length L Ch R = 1 ,25432   ,146,146,146
BEGIN DESCRIPTION:
Mapping XS 3ae1e4ff
END DESCRIPTION:
XS GIS Cut Line= 3
      2283940.08     13268246.28      2284114.55     13268230.66
      2284514.01      13267912.9
#Sta/Elev= 30
  4632.2  227.69  4639.9  226.96    4670  226.17  4683.4  224.82  4690.1  225.13
  4700.1  223.98  4730.2  223.08  4740.3  221.91  4800.5  218.44  4806.5  217.51
  4854.9  216.26  4883.7  214.11  4904.5  213.87  4912.3  212.99    4919  213.65
  4976.6  213.71    4983  214.41  4997.5  213.66  5054.2  214.25  5090.4  214.65
  5168.9  217.83    5182  219.24  5196.1  219.81  5210.5  221.35  5224.9  222.08
  5245.9   224.2  5260.1  226.19  5274.6  227.15    5297  229.59  5317.8  230.68
#Mann= 3 , 0 , 0
  4632.2     .16       0    4983     .07       0  5054.2     .16       0
Bank Sta=4983,5054.2
XS Rating Curve= 0 ,0
Exp/Cntr=0.3,0.1

Type RM Length L Ch R = 1 ,25286   ,146,146,146
BEGIN DESCRIPTION:
Mapping XS f772d2bb
END DESCRIPTION:
XS GIS Cut Line= 4
      2283988.25     13268340.03      2284135.38      13268380.4
      2284481.73     13268100.45      2284561.17     13268005.38
#Sta/Elev= 30
  4638.3  224.07  4668.9  223.35  4789.5  214.85  4802.4  214.51  4808.8  215.05
  4816.8   214.4  4837.6  214.89    4852  213.92  4858.4  214.23  4866.3   213.4
  4872.8  213.82  4895.1  213.05  4915.9  213.44  4936.7  212.41  4944.7  208.98
  4951.1   208.7  4959.1   206.9  4973.5  204.87  5000.4  203.15    5051  205.62
  5064.7  207.59    5079  209.19  5093.4  212.09  5115.3  213.91  5229.3   217.9
  5264.7  220.96  5306.3  223.61  5320.7  225.17  5349.3  226.61  5360.1  226.51
#Mann= 4 ,-1 , 0
  4638.3     .16       0  4959.1     .07       0  5064.7     .16       0
  5360.1     .05       0
Bank Sta=4959.1,5064.7
XS Rating Curve= 0 ,0
Exp/Cntr=0.3,0.1

Type RM Length L Ch R = 1 ,25140   ,385,385,385
BEGIN DESCRIPTION:
PAISANO CREEK 41.0
END DESCRIPTION:
XS GIS Cut Line= 3
      2283986.94     13268752.79      2284535.12     13268199.41
      2284652.29     13268075.73
#Sta/Elev= 30
  4480.2  220.76  4520.3  218.08  4640.5  212.16  4711.2  211.18  4739.5  210.48
  4746.6  209.59  4774.9  209.13  4796.1   209.6  4852.7  208.73  4859.7   208.1
  4923.4  208.27  4937.5  207.94  4944.6  206.77  4951.7  207.72  4958.7  206.92
    4980  206.82  4993.8  205.09  5015.3   207.5  5022.4  206.77  5029.4  208.11
  5036.5   208.1  5043.6  209.38  5121.4  211.91  5220.4  216.21  5298.2  220.93
  5312.3  221.24  5404.2  227.33  5418.3  226.73  5425.3  228.33  5429.5  228.33
#Mann= 3 , 0 , 0
  4480.2      .1       0  4951.7     .07       0  5029.4      .1       0
Bank Sta=4951.7,5029.4
XS Rating Curve= 0 ,0
Exp/Cntr=0.3,0.1

Type RM Length L Ch R = 1 ,24755   ,446,446,446
BEGIN DESCRIPTION:
PAISANO CREEK 40.0
END DESCRIPTION:
XS GIS Cut Line= 3
      2284137.71     13268946.86      2284437.72     13268746.85
      2284737.72     13268646.85
#Sta/Elev= 30
  4660.1  220.98  4682.6  219.23  4696.2     219  4709.7  216.85  4724.7  216.19
  4739.7  214.98  4754.8  212.86  4768.3  212.21  4775.8  211.12  4796.8  210.33
  4811.8  208.75  4948.6  203.74  4956.1  202.51  4977.1  201.87  4984.4  200.72
  4987.6  201.22  5023.3  201.43  5031.2  202.91  5052.3  204.29  5115.5   206.1
  5199.9  210.19  5220.9  210.56  5231.5  211.58    5242  211.86  5263.1  214.16
  5284.2   215.2  5305.3  217.55  5315.8  217.95  5326.4  219.65  5336.9  220.42
#Mann= 3 , 0 , 0
  4660.1      .1       0  4948.6     .07       0  5031.2      .1       0
Bank Sta=4948.6,5031.2
XS Rating Curve= 0 ,0
Exp/Cntr=0.3,0.1

Type RM Length L Ch R = 1 ,24309   ,415,415,415
BEGIN DESCRIPTION:
PAISANO CREEK 39.0
END DESCRIPTION:
XS GIS Cut Line= 3
      2284237.75     13269296.84      2284537.72     13269196.85
      2284837.75     13268896.83
#Sta/Elev= 30
  4655.4  215.22    4658  215.22  4676.4  212.75    4687  211.87  4697.5  211.64
  4708.1  210.42  4718.6  210.28  4729.2  209.29  4750.2  208.52  4771.3  206.88
  4781.9  206.58  4834.6  203.18  4887.3   201.1  4897.8  200.38  4929.4  199.27
  4961.1  198.76    4969  198.09  4975.1  198.09  4999.6  195.13    5014  197.47
  5098.9  199.82  5141.3   201.9  5169.6  202.46  5219.1  205.17  5254.4  207.51
  5282.7  208.72  5339.3  211.99  5367.6  214.45  5392.3  217.33  5395.9  217.33
#Mann= 3 , 0 , 0
  4655.4      .1       0  4975.1     .07       0    5014      .1       0
Bank Sta=4975.1,5014
XS Rating Curve= 0 ,0
Exp/Cntr=0.3,0.1

Type RM Length L Ch R = 1 ,23894   ,296,296,296
BEGIN DESCRIPTION:
PAISANO CREEK 38.0
END DESCRIPTION:
XS GIS Cut Line= 3
      2284437.73     13269646.85      2284737.72     13269546.85
      2285037.73     13269246.84
#Sta/Elev= 30
  4658.3  205.03  4660.9  205.03  4679.4  203.26  4732.1  201.22  4742.6  200.41
  4774.2  199.34  4784.8  198.61  4826.9  196.71  4858.6  196.05  4869.1  195.28
  4921.8  193.37  4932.4   193.5  4942.9  193.07  4988.7  192.94  4999.8  192.47
  5002.6  191.97  5005.8  192.47  5016.9  193.32  5059.4  193.71  5115.9     195
  5144.2  196.05  5186.7  198.45  5229.1  201.35  5257.4  202.76  5271.5  203.03
  5356.4  208.17  5370.5  209.37  5384.6  210.03  5395.2  211.28  5398.8  211.28
#Mann= 3 , 0 , 0
  4658.3      .1       0  4932.4     .07       0  5016.9      .1       0
Bank Sta=4932.4,5016.9
XS Rating Curve= 0 ,0
Exp/Cntr=0.3,0.1

Type RM Length L Ch R = 1 ,23598   ,188,188,188
BEGIN DESCRIPTION:
PAISANO CREEK 37.0
END DESCRIPTION:
XS GIS Cut Line= 3
      2284359.25     13269786.02      2284806.25     13269864.14
      2285259.78     13269445.33
#Sta/Elev= 30
  4420.4  202.26  4439.2  202.61  4454.3  202.02  4508.8  201.69  4513.8   200.7
  4550.8  199.97  4611.7   197.5  4687.3  192.75  4713.2   192.2  4746.7  190.42
  4801.2  189.23  4860.7  189.32  4872.1   188.5  4880.3  189.31  4944.2  189.65
 4973.91  190.59  4986.3  190.06 5011.78  190.65  5064.6  189.04  5142.2  190.85
  5170.6  192.79  5177.4  192.57  5191.6  193.54  5213.1  193.95  5319.2  200.49
  5361.7  202.13  5396.8  204.93  5432.6  206.56  5467.7  209.29  5491.5  210.04
#Mann= 3 , 0 , 0
  4420.4     .16       0 4973.91     .07       0 5011.78     .16       0
#XS Ineff= 2 ,-1
 4732.71 4972.04190.6464 5014.59 5134.54190.7299
Permanent Ineff=
       F       F
Bank Sta=4973.91,5011.78
XS Rating Curve= 0 ,0
Exp/Cntr=0.3,0.1

Type RM Length L Ch R = 1 ,23410   ,393,393,393
BEGIN DESCRIPTION:
PAISANO CREEK 37.1
END DESCRIPTION:
XS GIS Cut Line= 3
      2284487.72     13270496.85      2285037.72     13269896.85
      2285287.69     13269596.89
#Sta/Elev= 30
  4201.8  212.83  4286.6  210.29    4294  209.13  4343.3     207  4371.7  203.55
    4577  193.63  4739.8  188.31  4817.5  187.13  4839.1  181.95  4845.9  182.66
  4852.9  186.71    4881  186.66  4888.4   182.5  4894.9  181.24  4909.4  182.06
  4916.8  184.56  4923.5  181.75  4937.7  181.79  4945.1  186.19  4973.5   186.6
 4975.57  185.22  4980.3   182.1  4987.7  182.66  4994.5  186.54  5008.6  187.18
  5164.8  188.41  5242.9  191.79  5335.3  197.62  5356.1  197.75  5406.2  201.37
#Mann= 3 , 0 , 0
  4201.8     .16       0 4975.57     .07       0  5008.6     .16       0
#XS Ineff= 2 ,-1
 4808.28 4857.62185.9954  4879.9 4962.75185.9621
Permanent Ineff=
       F       F
Bank Sta=4975.57,5008.6
XS Rating Curve= 0 ,0
Exp/Cntr=0.3,0.1

Type RM Length L Ch R = 1 ,23017   ,40,40,40
BEGIN DESCRIPTION:
PAISANO CREEK 36.0
END DESCRIPTION:
XS GIS Cut Line= 3
      2285087.69     13270246.87      2285337.72     13270096.85
       2285537.7     13269796.88
#Sta/Elev= 30
  4682.8  191.29  4791.7  188.06  4844.2  185.65    4850   186.1  4902.5  183.94
  4916.1  182.14  4923.8  182.32  4929.7  180.57  4951.1  180.41  4960.8  181.05
  4966.6  180.43  4971.5  181.77  4977.4  181.77  4978.9  180.32  4981.6  179.82
  4987.9  180.57  5002.9  181.15  5010.4   180.4    5069  180.36  5082.5  181.04
  5096.1  182.23  5111.1  184.69  5147.1  185.79  5154.7  186.79  5198.2  189.71
  5249.3  192.24  5262.8  193.88  5306.4   197.1  5312.4  198.16  5334.9  199.45
#Mann= 3 , 0 , 0
  4682.8      .1       0  4977.4     .07       0  5002.9      .1       0
Bank Sta=4977.4,5002.9
XS Rating Curve= 0 ,0
Exp/Cntr=0.3,0.1

Type RM Length L Ch R = 1 ,22977   ,81,81,81
BEGIN DESCRIPTION:
Mapping XS 31b1ab36
END DESCRIPTION:
XS GIS Cut Line= 4
       2285208.3     13270355.03      2285295.11     13270181.41
       2285353.7     13270129.33       2285583.2     13269906.33
#Sta/Elev= 30
    4686  187.38  4818.1  184.91  4849.2  186.89  4854.8  185.32  4862.8  187.69
  4906.6  186.45  4927.5  187.82    4935  186.16  4941.7  187.79  4958.5     186
  4970.2  187.61  5026.7  187.04  5033.8  186.62  5037.9   182.9  5040.6   182.4
  5043.9   182.9  5047.9  186.02    5055  184.35    5062  186.17  5069.2   183.3
  5076.1  186.41  5083.3  184.28  5090.3  185.85  5097.5  184.36  5104.4  186.85
  5118.6  186.91  5125.8  185.31  5132.7  187.24  5154.1  186.51  5278.5  194.68
#Mann= 3 , 0 , 0
    4686      .1       0  4927.5     .07       0  5026.7      .1       0
Bank Sta=4927.5,5026.7
XS Rating Curve= 0 ,0
Exp/Cntr=0.3,0.1

Type RM Length L Ch R = 1 ,22896   ,294,294,294
BEGIN DESCRIPTION:
Mapping XS 1afe7c45
END DESCRIPTION:
XS GIS Cut Line= 4
      2285258.19     13270361.57      2285438.34     13270170.56
      2285494.76     13270040.36      2285618.45     13269949.22
#Sta/Elev= 30
  4684.8  186.31  4793.9  184.65  4822.2  183.73  4871.6  183.16  4899.9  181.54
  4907.2  182.81  4928.2  181.59  4935.5  181.97  4942.4  181.24  4952.1  181.34
  4957.6   179.9  4963.1  180.18  4986.5  179.13    4995  179.52  5004.6  179.19
    5010  179.45  5016.5  178.58  5019.8  179.08  5027.7  179.24  5049.5  180.94
    5057  182.25  5088.5   184.3  5130.2   186.1  5143.1  187.25    5187  189.78
  5201.6  189.97  5207.8  190.95  5237.1  192.08  5240.7  192.95  5242.9  192.95
#Mann= 3 , 0 , 0
  4684.8      .1       0  4952.1     .07       0  5049.5      .1       0
Bank Sta=4952.1,5049.5
XS Rating Curve= 0 ,0
Exp/Cntr=0.3,0.1

Type RM Length L Ch R = 1 ,22602   ,428,428,428
BEGIN DESCRIPTION:
PAISANO CREEK 35.0
END DESCRIPTION:
XS GIS Cut Line= 3
       2285537.7     13270596.89      2285687.72     13270296.85
      2285737.72     13270046.86
#Sta/Elev= 30
  4671.3  188.29  4707.7  187.14  4716.1  186.31    4730  186.05  4746.8  184.98
  4791.5  183.41  4841.8  182.06  4872.6  181.92    4881  181.13  4886.6  181.48
  4903.3  181.38  4908.9  180.85  4939.7  179.95  4948.1  179.21  4953.6  179.48
    4976  178.35  4984.4  178.55  4992.8  178.05  4998.4  177.03  5009.3  177.06
  5016.7  176.16  5027.1  177.15  5047.5  180.02  5057.7   180.1  5067.9  181.17
  5098.5  181.42  5139.3  183.09  5149.5  183.92  5190.3  185.49  5261.7  189.33
#Mann= 3 , 0 , 0
  4671.3      .1       0  4953.6     .07       0  5047.5      .1       0
Bank Sta=4953.6,5047.5
XS Rating Curve= 0 ,0
Exp/Cntr=0.3,0.1

Type RM Length L Ch R = 1 ,22174   ,606,606,606
BEGIN DESCRIPTION:
PAISANO CREEK 34.0
END DESCRIPTION:
XS GIS Cut Line= 3
      2286387.72     13270646.85      2286087.72     13270346.85
      2285887.73     13270046.87
#Sta/Elev= 30
  4589.4  191.04  4617.7  190.08    4646  188.55  4702.5  186.78  4773.2  183.92
  4829.8  181.52  4872.2  179.28  4914.7   178.4  4942.9  177.08  4957.1  177.02
  4971.2  176.18  5007.1  175.51  5009.9  175.01  5021.2  176.16  5049.7  176.83
  5057.2  176.67  5072.3  177.19  5099.3  177.95  5129.3  178.38  5186.4  180.54
  5201.4  180.81  5216.5   181.6    5230  181.76  5243.5   182.5  5273.6  183.46
  5302.1  185.01  5324.6  185.73  5345.7  187.08  5360.7  187.47  5374.2  188.27
#Mann= 3 , 0 , 0
  4589.4      .1       0  4957.1     .07       0  5072.3      .1       0
Bank Sta=4957.1,5072.3
XS Rating Curve= 0 ,0
Exp/Cntr=0.3,0.1

Type RM Length L Ch R = 1 ,21568   ,86,86,86
BEGIN DESCRIPTION:
PAISANO CREEK 33.0
END DESCRIPTION:
XS GIS Cut Line= 4
      2286537.72     13270396.89      2286525.58     13270118.48
      2286551.62     13270031.68      2286436.61     13269476.15
#Sta/Elev= 30
  4574.7  184.18  4614.8  183.39  4634.8  181.95  4754.9  177.68  4896.8  174.41
  4907.3  173.92  4912.8  172.86    4918  173.85  4928.2  172.21  4938.6  171.49
  4943.9  170.17  4991.4  167.72  5017.4  167.53  5020.2  167.03  5023.4  167.53
  5136.9  169.94  5173.6  172.52  5181.9  174.11  5187.1   173.9  5204.2  175.67
  5237.2  176.78  5265.5  179.51  5326.8  182.51  5332.5  183.35  5408.5  186.45
  5418.7  187.32  5432.9  187.51    5478  190.09  5483.1  189.62  5511.3  191.01
#Mann= 4 ,-1 , 0
  4574.7     .05       0    4918    .035       0  5181.9     .05       0
  5511.3     .05       0
Bank Sta=4918,5181.9
XS Rating Curve= 0 ,0
Exp/Cntr=0.3,0.1

Type RM Length L Ch R = 1 ,21482   ,94,94,94
BEGIN DESCRIPTION:
Mapping XS 3d2ffe63
END DESCRIPTION:
XS GIS Cut Line= 6
      2286590.68     13270411.41      2286573.32     13270135.84
      2286621.07      13269986.1      2286610.21     13269894.96
      2286566.81     13269773.43      2286527.95     13269460.34
#Sta/Elev= 30
  4605.8  184.15  4660.5  183.33  4760.7  179.17  4820.8   177.6  4850.8  177.89
  4870.9  177.24  4878.6  176.48  4881.9  176.98    4910  177.48  4942.2   177.7
  4947.4  177.19  4974.4  177.97  5068.5  178.35  5088.7  178.45  5106.7  179.47
  5111.8  178.57  5127.4   179.6  5210.6  179.06  5215.9  179.55  5306.8  179.12
  5337.1  180.91  5347.1  182.04  5397.5  184.44  5427.8  187.31  5454.2  189.15
  5459.3  188.92  5468.1  189.77  5528.5  193.11  5540.1  193.29  5575.4  195.58
#Mann= 4 ,-1 , 0
  4605.8     .05       0  4974.4    .035       0  5068.5     .05       0
  5575.4      .1       0
Bank Sta=4974.4,5068.5
XS Rating Curve= 0 ,0
Exp/Cntr=0.3,0.1

Type RM Length L Ch R = 1 ,21388   ,566,566,566
BEGIN DESCRIPTION:
PAISANO CREEK 32.0
END DESCRIPTION:
XS GIS Cut Line= 4
      2286655.79     13270483.07      2286668.81     13270140.18
      2286714.38     13269953.55       2286640.6     13269482.64
#Sta/Elev= 30
  4596.7  184.69    4653  183.29  4783.7   178.5  4893.1  176.02  4933.2  174.31
    4939  173.38  4952.4  172.96  4957.5  171.82    4994  170.75  4998.9  169.75
    5005  170.38  5056.5   171.7  5131.9  174.63  5205.9  171.82  5268.6  171.39
  5273.6  172.12  5300.7  172.89  5351.3  177.06  5391.8  179.35    5399  180.36
    5412  180.44  5432.3  182.42  5466.7  184.52  5503.1  188.44  5523.4  189.36
  5543.6  191.38  5553.7   191.5    5592  194.55  5597.1  194.13  5608.6   194.7
#Mann= 4 ,-1 , 0
  4596.7     .05       0  4957.5     .03       0  5056.5     .05       0
  5608.6      .1       0
Bank Sta=4957.5,5056.5
XS Rating Curve= 0 ,0
Exp/Cntr=0.3,0.1

Type RM Length L Ch R = 1 ,20822   ,418,418,418
BEGIN DESCRIPTION:
PAISANO CREEK 31.0
END DESCRIPTION:
XS GIS Cut Line= 3
       2286937.7     13270696.89      2287187.72     13270296.85
       2287437.7     13269896.89
#Sta/Elev= 30
  4491.4  190.72  4550.4  186.34  4556.9  185.36  4578.1  184.67  4608.8  181.67
  4635.9  180.07  4644.7  179.02  4703.1  175.91  4715.5  174.75  4809.8  170.09
  4897.7  166.53  4955.5  165.01  4960.2  164.01    4992  162.77  5007.4  163.03
    5013   162.1  5028.6  162.76  5034.5  164.45  5043.9  164.52  5049.8  165.61
  5065.1  166.23    5071  168.29  5101.7  169.26  5107.6  170.43  5174.8  170.99
  5201.9  172.44  5217.3  172.17    5275  173.53  5363.5  176.63  5434.8  179.89
#Mann= 3 , 0 , 0
  4491.4     .05       0  4955.5     .03       0  5034.5     .05       0
Bank Sta=4955.5,5034.5
XS Rating Curve= 0 ,0
Exp/Cntr=0.3,0.1

Type RM Length L Ch R = 1 ,20404   ,413,413,413
BEGIN DESCRIPTION:
PAISANO CREEK 30.0
END DESCRIPTION:
XS GIS Cut Line= 3
      2287237.75     13270846.82      2287487.72     13270546.85
      2287537.72     13269746.88
#Sta/Elev= 30
  4627.4  191.28  4691.8  186.63  4762.1  180.09  4811.5  176.95  4825.9  175.16
    4848   173.8  4854.5  172.63  4883.1  171.19  4918.3  168.41  4939.8  166.01
  4946.9  164.51  4967.7  163.45  4989.9  162.04  5010.7  161.95  5014.4  161.27
  5047.9  162.13  5057.9  163.23  5095.5  164.89  5168.2  166.57  5208.2  168.96
  5255.8  170.17  5338.5  169.26  5398.6  169.91  5416.1  171.63  5468.7   172.6
    5589  176.76  5629.1  179.13  5699.2  181.86  5789.4  186.99  5819.4  187.96
#Mann= 4 ,-1 , 0
  4627.4     .05       0  4967.7     .03       0  5057.9     .05       0
  5819.4     .05       0
Bank Sta=4967.7,5057.9
XS Rating Curve= 0 ,0
Exp/Cntr=0.3,0.1

Type RM Length L Ch R = 1 ,19991   ,421,421,421
BEGIN DESCRIPTION:
PAISANO CREEK 29.0
END DESCRIPTION:
XS GIS Cut Line= 3
      2287937.72     13271146.84      2287837.72     13270746.85
      2288037.72     13270246.86
#Sta/Elev= 30
  4589.1  181.38  4640.6  178.04  4653.5  177.71  4681.9  175.34  4694.7  175.01
  4730.8  172.06  4784.9  169.27  4813.3  167.14  4846.8  165.83    4888  162.37
  4895.7  161.22  4900.9   161.3  4918.9  159.79    4937  158.57  4949.9   158.8
  4978.2  157.82  4983.4  158.19  4998.6  156.43  5010.8  157.74  5040.4  159.86
  5055.2  161.74  5064.7  162.33  5070.1  162.14  5094.3   163.9  5109.1  163.97
  5141.4  165.56  5231.6  165.45  5315.1   166.3  5417.4  169.71  5539.9  173.05
#Mann= 3 , 0 , 0
  4589.1     .05       0  4918.9     .03       0  5040.4     .05       0
Bank Sta=4918.9,5040.4
XS Rating Curve= 0 ,0
Exp/Cntr=0.3,0.1

Type RM Length L Ch R = 1 ,19570   ,418,418,418
BEGIN DESCRIPTION:
PAISANO CREEK 28.0
END DESCRIPTION:
XS GIS Cut Line= 3
      2288087.73     13271146.82      2288237.72     13270796.85
      2288137.71     13270296.81
#Sta/Elev= 30
    4610  180.22  4664.4  176.04  4740.5  171.36  4747.8  170.49  4776.8  169.15
  4805.8  167.05  4838.4  165.37  4892.8  160.09  4905.5   159.7  4914.6  158.59
  4923.7  158.12  4929.1  158.42  4936.4  157.53  4958.1  156.98    4969  156.73
  4976.2  155.96  4981.7  156.11    4988  155.34  5008.1  154.83  5010.9  154.33
  5031.5  156.48  5051.9   157.4  5062.1  157.63  5072.3  158.44  5102.9  158.75
  5164.1  160.36  5174.3  161.22  5276.3  164.63  5357.9  166.17  5500.7  170.66
#Mann= 3 , 0 , 0
    4610     .05       0  4958.1    .035       0  5051.9     .05       0
Bank Sta=4958.1,5051.9
XS Rating Curve= 0 ,0
Exp/Cntr=0.3,0.1

Type RM Length L Ch R = 1 ,19152   ,402,402,402
BEGIN DESCRIPTION:
PAISANO CREEK 27.0
END DESCRIPTION:
XS GIS Cut Line= 3
      2288787.71     13270846.84      2288537.72     13270496.85
      2288237.73     13270246.86
#Sta/Elev= 30
  4591.4  180.58  4613.5  180.46  4628.3  179.43  4640.5  178.25  4649.1   176.6
    4670  176.14  4677.4  175.06  4690.9  174.24  4699.5  172.51  4714.3  171.36
  4726.6  169.74  4776.9  166.02  4791.7  165.46  4821.2  163.05    4863  160.92
  4886.3   159.4  4913.4  156.92    4949  154.93  4957.6  153.58  4972.3  152.72
  4984.4  151.42  4987.6  151.92  5024.8  153.38  5035.2  154.57  5099.6  158.55
  5199.2  162.02  5205.7  162.65  5283.8  165.51  5298.1  166.44    5412  170.47
#Mann= 3 , 0 , 0
  4591.4     .05       0    4949    .035       0  5035.2     .05       0
Bank Sta=4949,5035.2
XS Rating Curve= 0 ,0
Exp/Cntr=0.3,0.1

Type RM Length L Ch R = 1 ,18750   ,441,441,441
BEGIN DESCRIPTION:
PAISANO CREEK 26.0
END DESCRIPTION:
XS GIS Cut Line= 3
      2289087.73     13270696.87      2288887.72     13270296.85
      2288537.75     13270096.87
#Sta/Elev= 30
    4558  178.03  4580.4  176.44  4594.3  175.88  4647.5  171.88  4655.8  171.69
  4678.2  169.31  4692.2  168.83  4722.9  166.45  4736.9  165.83  4750.9  164.54
  4952.1   153.7  4968.9  151.86  4982.9   150.5  4993.8     150  4996.6   149.5
  5002.4  150.13  5018.9  150.38  5040.5  151.95  5072.2   153.1  5085.8  153.84
  5093.8  154.72  5108.9  154.95  5121.1   155.8  5174.4   157.5  5239.2  160.96
  5282.4  162.46  5298.2  163.61  5350.8  165.37  5357.2  166.09  5408.3     168
#Mann= 4 ,-1 , 0
    4558     .05       0  4968.9     .03       0  5040.5     .05       0
  5408.3     .05       0
Bank Sta=4968.9,5040.5
XS Rating Curve= 0 ,0
Exp/Cntr=0.3,0.1

Type RM Length L Ch R = 1 ,18309   ,278,278,278
BEGIN DESCRIPTION:
PAISANO CREEK 25.0
END DESCRIPTION:
XS GIS Cut Line= 3
      2289437.76     13270196.89      2289137.72     13269946.85
      2288787.69     13269846.85
#Sta/Elev= 30
  4618.2  172.05  4631.9  171.29  4639.7  170.31  4646.2  170.28  4668.4  168.33
  4746.5  164.44  4788.1  161.58  4802.4   161.2  4852.6  158.55  4859.7  157.56
  4902.7  155.38    4917  153.85  4930.7  153.37  4958.6  151.04  4966.5   149.5
  4987.3  147.93  5001.6  147.79  5005.3  147.24  5025.7  149.19  5071.2  150.72
  5098.5  151.24  5112.8  152.05  5123.2  151.86  5185.6  155.23  5210.3  155.67
  5216.8  156.62  5268.8  159.06  5283.1  159.34  5322.1  161.69  5372.8  163.64
#Mann= 4 ,-1 , 0
  4618.2     .05       0  4958.6     .03       0  5071.2     .05       0
  5372.8     .05       0
Bank Sta=4958.6,5071.2
XS Rating Curve= 0 ,0
Exp/Cntr=0.3,0.1

Type RM Length L Ch R = 1 ,18031   ,231,231,231
BEGIN DESCRIPTION:
PAISANO CREEK 24.0
END DESCRIPTION:
XS GIS Cut Line= 3
      2289575.43     13269929.92      2289371.44     13269782.35
      2288902.68     13269487.21
#Sta/Elev= 30
  4565.9  171.96  4601.5  169.66    4610  169.58  4616.2  168.81  4630.9  168.33
  4637.1  167.48  4651.8  167.08  4716.8  162.88  4773.2   159.9  4787.9  158.66
  4816.9  157.64  4832.7   156.2  4869.2  154.55  4948.1  149.41    4954   147.7
  4984.6  144.43  4990.2  143.26  5005.8  145.27  5021.1   145.3    5027  144.77
  5034.8  146.44  5048.2  147.04  5057.5  148.78  5063.5  148.69  5078.7  150.76
  5136.4  153.61  5194.1  155.16  5230.6  157.12  5251.8  157.63  5371.6  163.37
#Mann= 4 ,-1 , 0
  4565.9     .05       0  4948.1    .035       0  5078.7     .05       0
  5371.6     .05       0
Bank Sta=4948.1,5078.7
XS Rating Curve= 0 ,0
Exp/Cntr=0.3,0.1

Type RM Length L Ch R = 1 ,17800   ,208,208,208
BEGIN DESCRIPTION:
Mapping XS 9a0f8f21
END DESCRIPTION:
XS GIS Cut Line= 3
      2289705.66     13269773.69      2289128.38     13269348.33
      2288946.12      13269213.8
#Sta/Elev= 30
  4488.3  171.86  4512.5   170.2  4527.2   169.9  4535.4     169  4577.3  167.09
  4585.1  166.27  4648.3  163.25  4656.7   162.2  4662.9  162.26  4671.3  161.04
  4706.8  159.85    4784  155.68  4798.7  154.45  4813.3  154.16  4842.6  151.24
  4920.5  148.69  4928.2  147.81  4949.1  147.49  4975.3  146.46  4978.1  145.96
  4984.5  146.78  5013.8  146.87  5057.1  148.89    5064  148.77  5106.8   151.2
  5235.2  156.41  5314.6  160.44  5335.4  160.95  5414.8  164.71  5431.9  164.99
#Mann= 3 , 0 , 0
  4488.3     .05       0  4920.5    .035       0  5057.1     .05       0
Bank Sta=4920.5,5057.1
XS Rating Curve= 0 ,0
Exp/Cntr=0.3,0.1

Type RM Length L Ch R = 1 ,17592   ,285,285,285
BEGIN DESCRIPTION:
Mapping XS e13ce380
END DESCRIPTION:
XS GIS Cut Line= 4
      2289866.26     13269656.51      2289549.39     13269383.05
      2289215.19     13269179.06      2288981.75     13269166.09
#Sta/Elev= 30
  4419.1  174.02  4580.8  165.26  4621.9  163.98  4630.2  163.08  4687.2  160.37
  4744.2  158.51  4772.7  156.96    4787  155.45  4793.6  155.48  4822.1  152.54
  4842.7  151.49  4858.2  149.36  4879.5  148.29  4916.2  147.82  4922.1  146.63
  4931.7  146.96  4937.6  145.97    4953  145.59  4968.5  144.15  4989.8  143.69
  4995.4  142.98  5038.8  145.71  5097.4  147.71  5111.8  147.92  5185.3  151.41
  5229.2  152.69  5256.7  154.53  5286.8  155.46  5386.9  160.53    5463  163.48
#Mann= 3 , 0 , 0
  4419.1     .05       0  4916.2    .035       0  5097.4     .05       0
Bank Sta=4916.2,5097.4
XS Rating Curve= 0 ,0
Exp/Cntr=0.3,0.1

Type RM Length L Ch R = 1 ,17307   ,75,75,75
BEGIN DESCRIPTION:
PAISANO CREEK 23.0
END DESCRIPTION:
XS GIS Cut Line= 4
      2289627.72     13269390.01      2289589.53     13269117.47
      2289454.11     13268928.23      2289264.86     13268603.56
#Sta/Elev= 30
  4638.3  156.74  4772.8  151.95  4813.1  148.18  4818.3  146.97  4833.3  146.41
  4894.7  141.84  4937.5  139.58  4943.7  138.55  4994.1  136.87  5020.5  136.69
  5023.3  136.19  5029.7  137.02  5044.4  137.33  5080.1  137.06  5100.9  139.06
  5109.5   142.8  5115.7  143.18  5123.3  144.84  5130.4  147.44  5151.3  150.26
  5159.4  153.59    5167  154.41  5182.5   152.9  5188.5  150.38    5210  149.26
  5231.5  149.95  5262.9  152.18  5298.3  152.69  5327.4  153.96    5522  159.21
#Mann= 3 , 0 , 0
  4638.3     .05       0  4813.1    .035       0  5130.4     .05       0
Bank Sta=4813.1,5130.4
XS Rating Curve= 0 ,0
Exp/Cntr=0.3,0.1

Type RM Length L Ch R = 1 ,17232   ,98,98,98
BEGIN DESCRIPTION:
Mapping XS 4ab214a0
END DESCRIPTION:
XS GIS Cut Line= 5
       2289698.9     13269365.74       2289674.6     13269169.55
      2289645.08     13269072.33       2289554.8     13268940.38
      2289315.21     13268546.27
#Sta/Elev= 30
    4607  158.22    4747  152.87  4807.9  153.22  4811.9  151.84  4844.8  153.08
  4850.1  151.35  4870.2  152.18  4877.7  153.76  4882.9  150.71  4908.7  153.92
  4914.7   152.7  4923.6  153.86  4929.6  151.46  4944.6  153.86  4959.5  153.82
  4965.5  151.11  4973.5  153.32  4995.4  154.01  5001.4   151.6  5016.3     154
  5031.2  154.01  5037.3   151.9  5046.2  153.92  5052.2  150.29  5068.2  153.82
  5117.1  153.06  5175.4     149  5241.7  152.52  5437.4  157.93  5527.4  162.26
#Mann= 3 , 0 , 0
    4607     .05       0  4995.4    .035       0  5068.2     .05       0
Bank Sta=4995.4,5068.2
XS Rating Curve= 0 ,0
Exp/Cntr=0.3,0.1

Type RM Length L Ch R = 1 ,17134   ,692,692,692
BEGIN DESCRIPTION:
PAISANO CREEK 22.0
END DESCRIPTION:
XS GIS Cut Line= 2
      2289884.64     13269249.38      2289386.39     13268521.96
#Sta/Elev= 30
  4612.6  160.07  4792.2  149.87  4798.2  146.98  4807.1  146.58  4813.2  140.12
  4827.8  138.63    4843  140.03    4849  143.87  4863.9  144.93  4920.8  141.59
  4935.7  141.34  5001.4  139.73  5015.7  139.68  5028.4     141  5073.1  146.75
  5088.1  147.41  5094.1   148.7  5100.5  151.41    5109  152.17  5115.1     152
  5123.9  150.06  5136.9  148.97  5159.8  148.59  5180.8  149.24  5209.6  151.41
  5282.3  152.69  5345.3  154.97  5439.9  158.96  5476.2  161.71  5494.3  161.96
#Mann= 3 , 0 , 0
  4612.6     .05       0  4935.7    .035       0  5028.4     .05       0
Bank Sta=4935.7,5028.4
XS Rating Curve= 0 ,0
Exp/Cntr=0.3,0.1

Type RM Length L Ch R = 1 ,16442   ,434,434,434
BEGIN DESCRIPTION:
PAISANO CREEK 21.0
END DESCRIPTION:
XS GIS Cut Line= 3
       2290237.7     13268496.84      2290037.72     13268396.85
      2289787.76     13268296.87
#Sta/Elev= 30
  4779.9  151.61  4869.3  146.07  4891.7  144.35  4900.1   143.4    4914   142.8
  4922.4  141.36  4936.4  141.15  4981.1  137.78  4989.5  135.34  5000.4  133.52
  5006.2  134.02  5012.9  135.12  5018.3  135.36  5035.8  137.99  5042.5  138.77
  5047.9     139  5066.8  139.45  5072.1  139.19  5101.8  140.22  5111.2     141
  5120.6  141.27    5126  141.62  5132.7  142.55  5143.5  142.83  5150.2  143.58
    5165     144  5197.3  146.43  5233.7  148.51  5240.4  149.47  5272.7  151.56
#Mann= 3 , 0 , 0
  4779.9     .05       0  4981.1    .035       0  5035.8     .05       0
Bank Sta=4981.1,5035.8
XS Rating Curve= 0 ,0
Exp/Cntr=0.3,0.1

Type RM Length L Ch R = 1 ,16008   ,497,497,497
BEGIN DESCRIPTION:
PAISANO CREEK 20.0
END DESCRIPTION:
XS GIS Cut Line= 3
      2290337.74     13268246.89      2290187.72     13267996.85
       2289837.7     13267846.85
#Sta/Elev= 30
  4706.8  148.18  4751.5  146.72  4815.7  143.13  4846.8  142.06  4858.4  140.96
  4889.5   139.6  4940.1  136.31  4975.1  135.57  4995.2  131.98  4998.5  132.48
  5012.9  132.73  5020.2  133.51    5031   135.7  5052.8  137.02    5060  137.96
  5074.5  138.27  5083.6  139.49  5096.3  140.45  5107.2  140.76  5141.6  143.02
  5150.7  144.23  5159.8  144.59  5172.5  146.11  5205.1  148.92  5259.5  153.12
  5270.4   154.6  5281.3  155.24  5288.5  156.41  5346.5  160.59  5379.2  164.02
#Mann= 3 , 0 , 0
  4706.8     .05       0  4975.1    .035       0    5031     .05       0
Bank Sta=4975.1,5031
XS Rating Curve= 0 ,0
Exp/Cntr=0.3,0.1

Type RM Length L Ch R = 1 ,15511   ,433,433,433
BEGIN DESCRIPTION:
PAISANO CREEK 19.0
END DESCRIPTION:
XS GIS Cut Line= 3
      2290687.74     13267996.89      2290537.72     13267646.85
      2290137.76     13267546.86
#Sta/Elev= 30
  4624.4  148.23  4686.1  145.37  4700.6  144.13  4791.3  140.44    4862  136.12
  4874.7  136.23  4885.6  135.15  4929.1  133.33  4943.6  133.55  4950.8  132.61
  4961.7  132.32  4972.6  130.91  4983.5  130.78  4990.7  129.33  5002.3  128.16
  5015.5  130.12  5028.4  131.01  5036.2  133.54  5064.5     134  5139.2   136.9
    5147  137.71  5201.1  139.06  5262.9  141.57  5270.7  142.47  5275.8  142.21
  5311.9  143.54  5324.8  144.79  5358.3  146.56  5399.5   150.7  5417.5   151.4
#Mann= 4 ,-1 , 0
  4624.4      .1       0  4943.6     .07       0  5036.2      .1       0
  5417.5     .05       0
Bank Sta=4943.6,5036.2
XS Rating Curve= 0 ,0
Exp/Cntr=0.3,0.1

Type RM Length L Ch R = 1 ,15078   ,438,438,438
BEGIN DESCRIPTION:
PAISANO CREEK 18.0
END DESCRIPTION:
XS GIS Cut Line= 3
      2291137.72     13267946.86      2290937.72     13267546.85
      2290837.73      13266746.9
#Sta/Elev= 30
  4566.4  148.05  4625.1  145.44  4641.9  143.44  4700.6  139.61  4731.3  136.33
  4798.4  132.45  4932.6  130.67  4960.5  131.56  4968.9  130.24  4982.9  128.19
  4991.3  125.99    5005  125.38  5008.2  125.88  5010.8  129.84  5033.8  132.44
  5056.4  133.23  5346.2  134.92  5507.4  140.51  5620.8  148.39  5678.8  154.99
  5696.4  157.79  5701.4   157.5    5709  159.44  5739.2  162.76  5759.4  166.96
  5769.5  167.98    5777  170.13  5809.8  175.44  5817.3  178.79  5819.8  178.79
#Mann= 4 ,-1 , 0
  4566.4      .1       0  4968.9     .07       0  5010.8      .1       0
  5819.8     .16       0
Bank Sta=4968.9,5010.8
XS Rating Curve= 0 ,0
Exp/Cntr=0.3,0.1

Type RM Length L Ch R = 1 ,14640   ,452,452,452
BEGIN DESCRIPTION:
PAISANO CREEK 17.0
END DESCRIPTION:
XS GIS Cut Line= 3
      2291237.73     13267896.83      2291387.72     13267546.85
      2291387.72     13267146.81
#Sta/Elev= 30
  4654.9  145.71  4763.7  139.96  4821.7  138.01  4861.6  135.87  4868.8  134.91
  4883.3  134.75  4892.4  133.75  4897.8     134  4905.1  132.85  4937.7  131.16
    4945  130.24  4950.4  131.07  4959.5  130.03  4968.6  127.57    4974   127.4
  4981.3  125.56  4992.1  124.07  5002.8  123.41  5021.2  126.51  5026.6  125.69
  5032.9  126.96  5045.7  127.66  5145.7     130  5205.7   128.7  5265.7  128.66
  5295.7  129.36  5365.7   133.8  5375.7  135.47  5405.7  138.24  5435.7  142.56
#Mann= 4 ,-1 , 0
  4654.9      .1       0    4974     .07       0  5045.7      .1       0
  5435.7     .16       0
Bank Sta=4974,5045.7
XS Rating Curve= 0 ,0
Exp/Cntr=0.3,0.1

Type RM Length L Ch R = 1 ,14188   ,359,359,359
BEGIN DESCRIPTION:
PAISANO CREEK 16.0
END DESCRIPTION:
XS GIS Cut Line= 3
       2291937.7     13267846.82      2291687.72     13267246.85
      2291637.72     13267046.87
#Sta/Elev= 30
    4368  142.41  4530.5  137.95  4613.3  137.05  4725.5  137.71  4748.7   137.2
  4833.8  131.88  4866.3  130.65  4873.3  129.77  4920.5  128.03  4926.4  127.16
  4931.8  127.75  4942.1  126.17  4974.1  126.14  4985.5  124.91  5003.1  121.57
  5008.7  122.59  5015.2     125  5028.3  126.06  5069.5  128.89  5110.7  133.72
  5118.5  135.54  5131.3  136.45  5141.7  138.82    5152  139.55  5159.7  141.22
  5164.8  141.26  5200.9  147.69  5213.8   148.6  5221.5  150.49  5224.1  150.49
#Mann= 4 ,-1 , 0
    4368     .12       0  4974.1     .07       0  5028.3     .12       0
  5224.1      .1       0
Bank Sta=4974.1,5028.3
XS Rating Curve= 0 ,0
Exp/Cntr=0.3,0.1

Type RM Length L Ch R = 1 ,13829   ,493,493,493
BEGIN DESCRIPTION:
PAISANO CREEK 15.0
END DESCRIPTION:
XS GIS Cut Line= 3
      2291973.82     13267844.36      2292049.34     13267120.42
      2291831.68     13266959.76
#Sta/Elev= 30
  4421.5  142.49  4529.6   138.3  4630.1  135.46  4702.8  132.41  4730.7  134.02
    4791  134.21  4861.4  130.03  4921.7   125.6    4982  124.44  4990.1  119.56
  4992.9  119.06  5012.2  122.46  5052.4  125.18  5062.5   127.3  5112.7  131.52
  5148.6  136.07  5160.7  136.68  5166.9  137.76  5196.2  139.27    5217  141.14
  5225.4  140.98  5231.7  142.34  5246.3  141.92  5260.9   142.8  5267.1  143.86
    5311  146.18  5325.4  147.82  5367.4  150.31  5375.1  151.47  5419.9  152.73
#Mann= 4 ,-1 , 0
  4421.5     .12       0    4982     .07       0  5052.4     .12       0
  5419.9      .1       0
Bank Sta=4982,5052.4
XS Rating Curve= 0 ,0
Exp/Cntr=0.3,0.1

Type RM Length L Ch R = 1 ,13336   ,422,422,422
BEGIN DESCRIPTION:
PAISANO CREEK 14.0
END DESCRIPTION:
XS GIS Cut Line= 3
      2291937.73     13267996.85      2292537.72     13267296.85
      2292837.71     13266596.87
#Sta/Elev= 30
  4104.4  144.29  4224.6  142.38  4359.6  137.08    4466  131.44  4523.1  129.86
  4586.8   129.2  4650.4  130.64  4721.8  128.48  4742.6     129  4771.2  126.61
  4863.4  123.44  4934.1  122.77  4941.3   120.6  4947.9   122.9  4962.1  122.61
  4976.4  118.83  4990.4  117.02    5023  122.28  5048.1  124.09  5111.6  122.46
  5164.2  124.29  5245.7  123.88    5331  127.02  5407.1   128.2  5550.4  134.07
    5690   141.5  5702.7  141.96  5720.8  140.68  5726.3  142.13  5787.9   143.7
#Mann= 4 ,-1 , 0
  4104.4     .12       0  4962.1     .07       0    5023     .12       0
  5787.9      .1       0
#XS Ineff= 1 ,-1
 5047.66 5168.59  124.31
Permanent Ineff=
       F
Bank Sta=4962.1,5023
XS Rating Curve= 0 ,0
Exp/Cntr=0.3,0.1

Type RM Length L Ch R = 1 ,12914   ,401,401,401
BEGIN DESCRIPTION:
PAISANO CREEK 13.0
END DESCRIPTION:
XS GIS Cut Line= 3
      2292687.71     13267996.88      2292887.72     13267546.85
      2292987.71      13266946.9
#Sta/Elev= 30
  4470.2  142.29  4559.8  138.51  4577.6  136.39  4590.6  135.84  4600.9  136.49
  4623.4  135.41    4711   129.5  4743.8  128.41  4756.8  126.95  4855.3  121.53
    4908  120.58  4948.3  121.37  4965.2  120.63  4982.9  118.42  4995.4  115.33
  5003.2  117.87  5023.5  122.03  5056.4  120.22  5084.3  120.66  5094.5  121.87
    5135  123.82  5165.4   126.7  5178.1   129.1  5195.8   130.8  5276.9  131.42
  5299.8  132.89  5360.6  133.02  5510.1  137.18  5520.3  138.22  5570.9   138.2
#Mann= 4 ,-1 , 0
  4470.2     .12       0  4965.2     .07       0  5023.5     .12       0
  5570.9      .1       0
Bank Sta=4965.2,5023.5
XS Rating Curve= 0 ,0
Exp/Cntr=0.3,0.1

Type RM Length L Ch R = 1 ,12513   ,404,404,404
BEGIN DESCRIPTION:
PAISANO CREEK 12.0
END DESCRIPTION:
XS GIS Cut Line= 3
      2292887.76     13268046.82      2293187.72     13267796.85
      2293187.72     13266896.82
#Sta/Elev= 30
  4592.6  137.46  4677.8  134.05  4755.9  128.82  4762.4  129.58  4770.2  127.98
  4791.1  126.21  4840.5  123.73    4877  120.21  4932.9  118.87  4947.3   116.4
  4955.1  115.97  4961.6  116.82  4969.4  115.57  4975.9  116.76  4979.8  115.69
  5002.8   114.4  5023.1  118.32  5043.1  119.52  5083.1  120.27  5113.1  119.32
  5173.1  121.12  5183.1   121.5  5193.1  123.41  5263.1  126.02  5323.1  129.82
  5413.1  132.82  5633.1  132.49  5753.1  133.65  5773.1  134.58  5883.1  136.15
#Mann= 4 ,-1 , 0
  4592.6      .1       0  4932.9     .07       0  5043.1      .1       0
  5883.1      .1       0
Bank Sta=4932.9,5043.1
XS Rating Curve= 0 ,0
Exp/Cntr=0.3,0.1

Type RM Length L Ch R = 1 ,12109   ,418,418,418
BEGIN DESCRIPTION:
PAISANO CREEK 11.0
END DESCRIPTION:
XS GIS Cut Line= 3
      2292937.73     13268146.85      2293437.72     13268096.85
      2293737.72     13266596.85
#Sta/Elev= 30
  4496.4   137.6  4536.6  135.97  4586.8  132.91    4627  131.78  4677.3   128.3
  4757.7  124.88  4807.9  121.85  4838.1  120.92  4868.2  118.64  4908.4  117.75
  4938.6  118.57  4946.1  119.57  4958.7  119.92  4973.6  118.84  4978.8  117.99
  4996.1  112.29  5019.3  115.62  5029.5  118.94  5090.7  118.58  5121.3  117.67
  5172.3  119.73  5182.5  122.15  5274.2  126.33  5284.4   127.7    5417  131.23
  5743.3  132.49  6090.1  130.94  6161.5  131.29  6283.8  132.77  6528.6  140.65
#Mann= 4 ,-1 , 0
  4496.4      .1       0  4973.6     .07       0  5029.5      .1       0
  6528.6      .1       0
Bank Sta=4973.6,5029.5
XS Rating Curve= 0 ,0
Exp/Cntr=0.3,0.1

Type RM Length L Ch R = 1 ,11691   ,728,728,728
BEGIN DESCRIPTION:
PAISANO CREEK 10.0
END DESCRIPTION:
XS GIS Cut Line= 3
      2293087.69     13268596.86      2293687.72     13268446.85
      2293987.72     13266646.88
#Sta/Elev= 30
  4361.1  134.43  4443.6  130.83  4585.3  122.53  4649.7  120.91  4773.4  120.17
  4879.1  115.92  4969.3  118.46    4977  115.69  4982.1  115.69  5007.2  110.91
  5010.5  111.41  5020.1  117.17  5040.4  118.12    5081  116.15  5121.5  117.56
  5151.9  119.97  5182.4  121.11    5195  122.98  5316.7  128.85  5405.4  129.11
  5476.4  130.63  5859.1     130    5892  130.72  5993.4  129.65  6054.2   130.2
  6064.4  129.42  6533.2  130.68  6611.8  132.21  6632.1   133.4  6804.4  136.21
#Mann= 4 ,-1 , 0
  4361.1     .16       0  4969.3     .07       0  5040.4     .16       0
  6804.4     .05       0
Bank Sta=4969.3,5040.4
XS Rating Curve= 0 ,0
Exp/Cntr=0.3,0.1

Type RM Length L Ch R = 1 ,10963   ,1643,1643,1643
BEGIN DESCRIPTION:
PAISANO CREEK 9.0
END DESCRIPTION:
XS GIS Cut Line= 3
      2292837.76     13269946.83      2294459.25     13268760.47
      2294343.17     13266720.82
#Sta/Elev= 30
  3467.7  167.29  3481.2  165.71  3581.6  161.88  3918.2  150.42  4039.4  144.53
  4047.9  143.11  4062.4   143.3  4068.7  141.84  4089.6  141.91  4098.1  140.49
  4118.9  140.64  4125.1  139.41  4204.6  136.88  4254.8  133.99  4411.6  129.17
  4669.6   118.4  4798.4  116.45  4892.5  113.47  4984.4  116.68  4991.7     115
  5005.1  109.69    5020  115.12  5034.6  116.34    5064  114.54  5363.4  123.09
  5392.1  122.07  5400.6  123.25  5620.7  122.99  5961.2  126.32  7519.8  128.45
#Mann= 4 ,-1 , 0
  3467.7     .16       0  4984.4     .07       0  5034.6      .1       0
  7519.8      .1       0
Bank Sta=4984.4,5034.6
XS Rating Curve= 0 ,0
Exp/Cntr=0.3,0.1

Type RM Length L Ch R = 1 ,9320    ,571,571,571
BEGIN DESCRIPTION:
PAISANO CREEK 8.0
END DESCRIPTION:
XS GIS Cut Line= 3
      2293987.68     13270996.88      2295076.38     13270179.65
      2294487.71     13267396.83
#Sta/Elev= 30
    3853  152.32  3989.5  147.22  4474.8  122.81  4610.2  118.68  4831.1  115.05
  4916.5  111.24  4966.5  111.12    4981  108.35  5003.2  107.08  5010.2  107.72
  5024.8  111.41    5031  112.09  5116.4  111.75  5166.4  109.74  5203.5  109.75
  5268.3   111.2  5482.9   112.9  5758.6  111.69  5942.9  113.74  6188.2  114.69
  6280.2   115.6  6310.8  117.23  6331.3  116.66  6402.8  119.76    6489  121.61
  6515.3  123.62  6566.4  121.66  6876.5  122.61  7313.7  125.55  8058.7  126.76
#Mann= 4 ,-1 , 0
    3853     .05       0  4966.5    .035       0  5024.8     .05       0
  8058.7     .05       0
Bank Sta=4966.5,5024.8
XS Rating Curve= 0 ,0
Exp/Cntr=0.3,0.1

Type RM Length L Ch R = 1 ,8749    ,502,502,502
BEGIN DESCRIPTION:
PAISANO CREEK 7.0
END DESCRIPTION:
XS GIS Cut Line= 3
      2294287.68     13271096.87      2295545.13     13270471.31
      2294887.73     13267896.88
#Sta/Elev= 30
  3731.6  144.11  4120.8  123.08  4232.7   118.7  4401.8  116.19  4708.6  114.12
  4859.7  110.71  4870.9  109.49  4954.9  110.72  4960.5  109.35  4971.4  109.58
  4971.5  109.57  4993.7  105.36  4996.7  103.25  4999.5  102.75  5027.7   109.6
  5044.5  107.69  5072.5  110.28  5161.3  108.99  5243.9  110.38  5336.8  109.17
  5419.3  110.24  5748.2  108.02  6007.6  111.33  6115.9  113.57  6192.4  116.65
  6355.8  118.64  6771.4  120.74  6998.4   120.2  7514.5  124.44  7793.1     124
#Mann= 4 ,-1 , 0
  3731.6     .16       0  4971.4     .07       0  5027.7     .12       0
  7793.1     .05       0
Bank Sta=4971.5,5027.7
XS Rating Curve= 0 ,0
Exp/Cntr=0.3,0.1

Type RM Length L Ch R = 1 ,8247    ,908,908,908
BEGIN DESCRIPTION:
Mapping XS eaa094dc
END DESCRIPTION:
XS GIS Cut Line= 4
      2294528.34      13271771.2      2295678.51     13271109.31
      2295895.52     13270696.99      2295309.74     13268321.31
#Sta/Elev= 30
  3353.3  142.01  3721.8  123.48  3883.3  118.17  4358.3  114.93  4667.9  117.05
  4807.4  112.02  4821.3  109.79  4852.6  108.43  4865.3  103.64  4875.2  103.24
  4887.4  103.58  4909.4   107.7  4986.3  108.82  4999.5  102.81    5008  101.46
  5030.3  108.11  5367.3  109.29  5424.5   107.5  5496.9  108.71    5682  107.16
  5782.2  109.44  5939.5  109.77  5989.6  111.97  6011.6  110.94  6145.5  114.78
  6326.6  116.47  6414.7  115.14  6995.5  118.39  7493.3  118.85  7593.1  120.55
#Mann= 4 ,-1 , 0
  3353.3     .12       0  4986.3     .07       0  5030.3      .1       0
  7593.1     .16       0
Bank Sta=4986.3,5030.3
XS Rating Curve= 0 ,0
Exp/Cntr=0.3,0.1

Type RM Length L Ch R = 1 ,7339    ,350,350,350
BEGIN DESCRIPTION:
PAISANO CREEK 6.0
END DESCRIPTION:
XS GIS Cut Line= 3
       2295337.7     13272246.87      2296337.72     13271446.85
      2295737.72     13268746.86
#Sta/Elev= 30
    3677  120.33  3882.7  117.52  4089.2  116.54  4729.5  117.99  4801.6  116.33
  4822.4  113.04  4907.2  106.54  4921.6  103.97    4944  102.31  4954.4  100.04
  4976.6   98.79    4982  100.25  4998.6   99.54  5025.5  102.87  5049.8  103.71
  5244.5  106.09  5387.9  104.49  5491.6  104.69  5705.5  106.57  5736.2  108.27
  5828.4  107.45    6105  108.35  6166.4   107.3    6443  111.67  6636.4  113.44
  7097.3  114.02  7286.9  115.46  7416.2  115.16  7477.7  116.76  7723.5     117
#Mann= 4 ,-1 , 0
    3677     .05       0  4921.6    .035       0  5049.8     .05       0
  7723.5      .1       0
Bank Sta=4921.6,5049.8
XS Rating Curve= 0 ,0
Exp/Cntr=0.3,0.1

Type RM Length L Ch R = 1 ,6989    ,400,400,400
BEGIN DESCRIPTION:
Mapping XS ad98101e
END DESCRIPTION:
XS GIS Cut Line= 4
      2295777.89      13272222.6      2296548.73     13271673.98
      2296770.96     13271417.04      2296604.29     13269736.53
#Sta/Elev= 30
  3954.8  117.51  4224.6  117.11  4323.6   117.9  4676.5  118.11  4718.3   118.8
    4813  118.33  4884.3  114.62  4897.2  111.24  4900.9  111.24  4905.4  109.14
    4912  108.18  4919.6  105.27  4933.9  103.57  4940.5  103.65  4948.2  102.34
  4997.3   99.07    5026   101.1  5061.2  101.15  5110.5  103.19    5271  103.89
  5421.1  102.18  5542.3  104.07  5914.1  103.56  6265.8  104.17  6435.2  105.57
  6657.7  110.21  6758.2  111.13  6808.5  112.61  6828.6  111.85  6929.4  112.28
#Mann= 5 ,-1 , 0
  3954.8     .05       0  4940.5      .1       0  4940.5    .035       0
  5110.5     .05       0  6929.4      .1       0
Bank Sta=4940.5,5110.5
XS Rating Curve= 0 ,0
Exp/Cntr=0.3,0.1

Type RM Length L Ch R = 1 ,6589    ,922,922,922
BEGIN DESCRIPTION:
Mapping XS c47d2e2a
END DESCRIPTION:
XS GIS Cut Line= 4
      2296269.18     13272056.64      2296824.78     13271796.21
      2296937.62     13271744.12      2297649.44     13270303.14
#Sta/Elev= 30
  4099.5  117.79  4272.4  118.67  4285.6  118.13  4443.2  119.43  4550.7  118.29
  4580.1  117.15    4617  116.82  4625.8  116.09  4648.6   116.1  4856.7  108.33
  4923.6  104.68  4962.2  101.11  4979.1   98.98  5006.8   97.77  5012.8   99.49
  5035.1  101.45  5074.4  102.67  5124.9  102.08  5192.2   102.5    5247  101.21
  5304.4  100.91  5411.1  102.11  5626.2   101.2  5792.6  102.43    6045  101.75
  6073.1  101.09  6140.4  101.88  6185.3  103.49  6284.3  105.48  6444.6  111.19
#Mann= 3 , 0 , 0
  4099.5     .05       0  4962.2    .035       0  5035.1     .05       0
Bank Sta=4962.2,5035.1
XS Rating Curve= 0 ,0
Exp/Cntr=0.3,0.1

Type RM Length L Ch R = 1 ,5667    ,417,417,417
BEGIN DESCRIPTION:
Mapping XS 972e748e
END DESCRIPTION:
XS GIS Cut Line= 2
      2296625.14     13271993.42      2298847.33     13271139.27
#Sta/Elev= 30
  3618.6  118.57  3764.2  116.46  4067.4  105.41  4152.1  103.51    4382  101.57
  4671.3  101.15  4788.7   99.62    4794   98.31  4848.7    99.3    4854   97.48
  4878.7   97.01  4903.3   98.31  4908.7   96.53    4928   97.59  4933.3   96.69
    4958   97.03  4971.2   96.06  5127.1   94.91  5132.7   95.88    5152   95.46
  5157.3   96.99    5182   95.86  5187.3   97.54  5228.4   98.77  5281.9   95.64
  5326.6   98.77  5460.6  104.13  5667.6  110.58  5799.2  112.19  5999.3  112.85
#Mann= 5 ,-1 , 0
  3618.6      .1       0    4928     .05       0    4928     .07       0
  5187.3      .1       0  5999.3     .05       0
Bank Sta=4928,5187.3
XS Rating Curve= 0 ,0
Exp/Cntr=0.3,0.1

Type RM Length L Ch R = 1 ,5250    ,625,625,625
BEGIN DESCRIPTION:
PAISANO CREEK 5.0
END DESCRIPTION:
XS GIS Cut Line= 2
      2296703.93     13272119.79        2298771.     13271347.58
#Sta/Elev= 30
  3301.1  116.79  3322.5  115.66  3352.8  115.72  3383.1  114.79  3579.2  107.25
  3764.2  103.53  4092.5  100.61  4147.8   101.1  4208.4  100.32  4447.4  100.57
  4666.5   99.25  4812.7    99.8  4928.5   98.21  4938.4   99.33  4953.5   98.27
  4970.4   98.15  4978.5   97.19  4983.8   95.09  5002.2    92.7  5023.8   93.82
  5039.1   96.51  5055.8    97.4  5077.2  100.44  5087.9   101.1  5099.7  103.15
  5162.6  107.76    5248  110.46  5290.4  109.64  5356.3  111.31  5507.7  111.82
#Mann= 3 , 0 , 0
  3301.1      .1       0  4978.5     .07       0  5055.8      .1       0
Bank Sta=4978.5,5055.8
XS Rating Curve= 0 ,0
Exp/Cntr=0.3,0.1
