HEC-RAS study UNT003 IN NURI.prj: UNT003 IN NURI Base Level Engineering

--- UNT003 IN NURI.g01 (geometry) --- (continued)

Type RM Length L Ch R = 1 ,83779   ,395,395,395
BEGIN DESCRIPTION:
UNT003 IN NURI 124.0
END DESCRIPTION:
XS GIS Cut Line= 4
      2303192.67     13347479.12      2302755.71      13347640.1
      2301858.74     13348790.07       2301778.6     13349213.67
#Sta/Elev= 30
  3537.6  296.61  3585.5  295.17  3713.4  294.26  3804.9  290.56  4191.4   285.8
    4496  284.07  4743.6  282.47  4875.2  283.39  4947.5  281.23  5000.7  280.19
  5003.4  279.69  5006.7  280.19  5140.2  282.47  5151.2   282.8  5217.2  284.58
  5267.4  287.16    5275  288.45  5310.3  288.61  5395.4  292.27    5418  294.61
  5461.7  296.22  5488.9  299.32  5499.1  299.06  5539.8  301.81  5546.4  303.21
  5580.5  303.91  5603.8  306.24  5621.2  306.29  5682.3  310.47  5892.8  317.55
#Mann= 7 ,-1 , 0
  3537.6      .1       0    4496     .05       0  4743.6      .1       0
  4947.5     .05       0  5000.7     .03       0  5006.7     .05       0
  5151.2     .05       0
Bank Sta=4875.2,5140.2
XS Rating Curve= 0 ,0
Exp/Cntr=0.3,0.1

Type RM Length L Ch R = 1 ,83384   ,528,528,528
BEGIN DESCRIPTION:
UNT003 IN NURI 123.0
END DESCRIPTION:
XS GIS Cut Line= 4
      2302755.71     13347065.12      2302307.23     13347387.11
      2301571.25     13348675.08      2301513.75     13349227.07
#Sta/Elev= 30
    3366   294.9  3530.8  291.22  3818.1  289.38  4133.7  284.17  4494.7  282.32
  4661.1   282.3  4666.1  282.39  4840.8  281.54  4848.1  281.53  4898.6  281.16
    4936  277.92  4957.6  280.15  4992.1  277.29  4994.8  276.79  4998.1  277.29
  5010.9  279.61  5046.5  280.56  5071.7  282.12  5295.3  287.62  5360.7  288.89
  5473.7   295.6  5493.8  294.96  5624.5  303.61    5725  305.87  5765.3  310.29
  5771.8  309.15  5845.7  313.42  5885.7  313.74  5905.8  316.17  5956.5  318.09
#Mann= 13 ,-1 , 0
    3366      .1       0  4133.7     .05       0  4494.7      .1       0
  4661.1     .05       0  4666.1      .1       0  4840.8     .05       0
  4848.1     .12       0  4992.1     .07       0  4998.1     .12       0
  5071.7      .1       0  5295.3     .05       0  5885.7      .1       0
  5905.8     .05       0
Bank Sta=4957.6,5046.5
XS Rating Curve= 0 ,0
Exp/Cntr=0.3,0.1

Type RM Length L Ch R = 1 ,82856   ,60,60,60
BEGIN DESCRIPTION:
Mapping XS d5351c67
END DESCRIPTION:
XS GIS Cut Line= 3
      2302028.17     13346691.11      2301272.95     13348165.09
      2301158.36     13348761.49
#Sta/Elev= 30
  3445.4  300.51  3451.8  299.64  3750.1  292.17    3918  289.22  4045.6  285.32
    4201   282.9  4206.6  283.66  4245.4  282.26  4378.6   282.4  4451.9  283.59
  4484.3  282.64  4639.4  279.13  4804.1  280.52  4822.7  281.32  4922.4  280.08
  4944.6  278.23  4950.2  276.15  4999.5  276.02  5002.2  275.52  5005.5  276.02
    5039  276.18  5055.6   281.4  5090.1   281.8  5209.6  287.45  5276.8  289.08
    5307  289.78  5408.9  292.11  5439.4  293.78  5592.2  296.42  5708.9  299.83
#Mann= 9 ,-1 , 0
  3445.4     .05       0  3750.1      .1       0  4484.3     .05       0
  4804.1      .1       0  4999.5     .07       0  5005.5      .1       0
  5090.1     .05       0  5276.8      .1       0    5307     .05       0
Bank Sta=4922.4,5055.6
XS Rating Curve= 0 ,0
Exp/Cntr=0.3,0.1

Type RM Length L Ch R = 1 ,82796   ,69,69,69
BEGIN DESCRIPTION:
UNT003 IN NURI 122.0
END DESCRIPTION:
XS GIS Cut Line= 4
      2301993.07     13346673.28       2301323.3     13347988.88
      2301212.18     13348091.31      2301114.61     13348746.17
#Sta/Elev= 30
  3464.3  301.01  3777.6  292.54  3908.7  290.38    4170   283.9  4309.9  282.44
  4409.1  283.42  4453.6  281.99  4509.4  282.37  4637.1  279.49  4784.8  280.01
  4876.2  279.19  4898.4  277.65  4971.5  279.81  4975.3  276.83  4978.1  276.33
  4981.3  276.83  4985.7  279.42  4992.5  277.11  4999.9  279.81  5014.1  279.79
  5020.9     279  5091.3  280.31  5169.5  284.44  5233.7  286.25  5299.5  288.71
  5349.9  289.12  5552.3  294.42  5565.3  293.89    5714  296.85  5753.8  298.47
#Mann= 9 ,-1 , 0
  3464.3     .05       0  3777.6      .1       0  4509.4     .05       0
  4784.8      .1       0  4975.3     .07       0  4981.3      .1       0
  5169.5     .05       0  5233.7      .1       0  5349.9     .05       0
Bank Sta=4971.5,5014.1
XS Rating Curve= 0 ,0
Exp/Cntr=0.3,0.1

Type RM Length L Ch R = 1 ,82727   ,350,350,350
BEGIN DESCRIPTION:
Mapping XS d4d9f581
END DESCRIPTION:
XS GIS Cut Line= 4
      2301960.43     13346667.73      2301312.01     13347899.47
      2301155.76     13348063.53      2301049.09     13348742.55
#Sta/Elev= 30
  3510.1  301.17  3821.6  292.86  3983.8  289.94  3994.2  288.95  4186.8  284.67
    4319   283.2  4407.2  283.75    4546  281.74  4554.7  281.86    4667  279.65
  4768.9  279.75    4875  279.25  4880.6  279.99  4887.8  278.69  4924.6  276.74
  4959.8  277.67  4961.8  277.62  4985.2   276.5  4987.9     276  4991.2   276.5
  5037.5  277.81    5080  278.55  5122.4   280.9  5265.9   285.5  5314.2  287.05
  5395.1  287.84  5607.8   292.1  5617.9   291.3  5638.1  293.12    5816  297.12
#Mann= 11 ,-1 , 0
  3510.1     .05       0  3821.6      .1       0    4546     .05       0
  4554.7      .1       0    4667     .05       0  4768.9      .1       0
  4961.8     .05       0  4985.2     .03       0  4991.2     .05       0
  5265.9      .1       0  5395.1     .05       0
Bank Sta=4959.8,5037.5
XS Rating Curve= 0 ,0
Exp/Cntr=0.3,0.1

Type RM Length L Ch R = 1 ,82377   ,387,387,387
BEGIN DESCRIPTION:
UNT003 IN NURI 121.0
END DESCRIPTION:
XS GIS Cut Line= 3
      2301887.74     13346546.82      2300987.72     13347746.85
      2299787.71     13347946.86
#Sta/Elev= 30
  3534.4  304.02  3570.9   304.2  3591.7  303.48    3598  301.88  3677.1   299.3
  3706.3  298.73  3727.1  300.19  3741.7  298.67  4112.6  292.76    4299   288.1
  4706.3  281.74  4791.7  278.42  4834.4  278.64  4870.9  275.39  4906.3  275.55
  4924.1  273.73  4926.9  273.23  4930.1  273.73  4941.7  276.19  4962.6  276.48
    4998   273.8  5044.6  276.34  5214.7   279.7  5238.1  279.98  5355.3  281.38
  5422.7  282.58  5658.9  288.96  5804.9  291.09  5996.5  296.38    6251  306.09
#Mann= 10 ,-1 , 0
  3534.4      .1       0    4299     .05       0  4924.1     .03       0
  4930.1     .05       0  5214.7      .1       0  5238.1     .05       0
  5355.3      .1       0  5422.7     .05       0  5658.9      .1       0
  5996.5     .05       0
Bank Sta=4962.6,5044.6
XS Rating Curve= 0 ,0
Exp/Cntr=0.3,0.1

Type RM Length L Ch R = 1 ,81990   ,413,413,413
BEGIN DESCRIPTION:
UNT003 IN NURI 120.0
END DESCRIPTION:
XS GIS Cut Line= 3
      2301937.75     13346246.83      2300737.72     13347446.85
      2299637.69     13347846.87
#Sta/Elev= 30
  3338.3   309.5  3479.8  305.34  3493.9  306.01    3706  300.06  3734.3  300.21
  3861.6  295.56  4073.7  291.09    4201  286.36  4266.6   286.3  4328.3  283.37
  4413.1  281.25  4724.3  279.45  4809.1  276.92  4879.8  277.17  4936.4  274.15
  4978.8  274.58  5004.1  272.66  5006.9  272.16  5010.1  272.66  5031.9     275
    5076  275.74  5088.6  277.22  5100.2  277.61  5172.6  278.91  5354.6  280.44
  5459.3  283.33  5725.9  292.72  5822.8  296.81  6181.4  308.57  6205.9  309.79
#Mann= 9 ,-1 , 0
  3338.3      .1       0  4266.6     .05       0  5004.1     .03       0
  5010.1     .05       0  5100.2      .1       0  5172.6     .05       0
  5459.3      .1       0  5725.9     .05       0  6181.4      .1       0
Bank Sta=4879.8,5088.6
XS Rating Curve= 0 ,0
Exp/Cntr=0.3,0.1

Type RM Length L Ch R = 1 ,81577   ,351,351,351
BEGIN DESCRIPTION:
UNT003 IN NURI 119.0
END DESCRIPTION:
XS GIS Cut Line= 3
      2301260.77     13346651.12      2300087.79     13347352.61
      2299708.33     13347571.09
#Sta/Elev= 30
  4132.5  286.88  4174.9  286.57  4328.5   282.1  4428.9  280.92    4474   278.9
  4583.4  277.29  4795.4  276.13  4846.8  276.55  4859.6  275.35  4905.1  275.01
  4917.9  273.07  4933.5  271.97  4963.3  274.36  4976.3  273.84  4995.3  271.65
    4998  271.15  5001.3  271.65  5034.6  274.53  5056.6  276.48    5124  277.61
  5133.2   277.7  5220.1  279.66  5289.6  283.18    5305  282.74  5357.5   286.2
  5384.7  285.91  5474.6  289.12  5490.1  289.62  5697.2  295.79  5937.1  303.87
#Mann= 10 ,-1 , 0
  4132.5      .1       0  4428.9     .05       0  4995.3     .03       0
  5001.3     .05       0    5124      .1       0  5133.2     .05       0
  5220.1      .1       0  5474.6     .05       0  5490.1      .1       0
  5697.2     .05       0
Bank Sta=4963.3,5034.6
XS Rating Curve= 0 ,0
Exp/Cntr=0.3,0.1

Type RM Length L Ch R = 1 ,81226   ,551,551,551
BEGIN DESCRIPTION:
UNT003 IN NURI 118.0
END DESCRIPTION:
XS GIS Cut Line= 3
      2301122.79     13346363.64      2300858.27     13346386.64
       2299846.3     13347191.61
#Sta/Elev= 30
  4099.3  285.43    4255  281.69  4335.3  281.11  4529.5  277.41  4742.6   275.3
  4763.4  275.99  4840.2  275.21  4895.5  275.66    4914  275.42  4941.2   272.1
  4979.3  272.22  4991.6  271.52  4995.9  270.19  4998.6  269.69  5001.9  270.19
  5019.7  271.08  5027.7  272.75  5048.5  272.25  5055.5  273.78  5069.3  275.01
  5104.6  275.88    5127  276.22  5239.5  282.24  5404.1  288.07  5412.1  287.59
  5482.6   289.5  5517.8  289.27  5546.7  290.71  5584.2  290.56  5657.9  291.64
#Mann= 9 ,-1 , 0
  4099.3      .1       0  4840.2     .05       0  4895.5      .1       0
  4979.3     .05       0  4995.9    .035       0  5001.9     .05       0
  5104.6      .1       0  5239.5     .05       0  5584.2      .1       0
Bank Sta=4914,5069.3
XS Rating Curve= 0 ,0
Exp/Cntr=0.3,0.1

Type RM Length L Ch R = 1 ,80675   ,454,454,454
BEGIN DESCRIPTION:
UNT003 IN NURI 117.0
END DESCRIPTION:
XS GIS Cut Line= 3
      2301287.72     13345596.85      2300087.72     13346296.85
      2299487.71     13347496.87
#Sta/Elev= 30
  3592.7  296.93    4076   282.6  4359.7   278.8  4471.3  280.77  4477.1  281.81
  4551.5  282.01    4798  274.34  4909.6  272.73  4952.6  273.34  4958.8  271.27
  4968.3  270.19  4974.1  271.47  4990.3   270.9  4995.9  265.62  5001.3  265.37
  5004.1  264.87  5007.3  265.37  5012.7  265.67  5026.7   270.9  5071.4  273.36
  5130.1  276.45    5295  273.63  5398.4  274.02  5465.5  275.16  5638.8  281.02
  5689.1  281.12  5710.3  282.61  6024.5  293.05  6291.7  304.09  6323.6  305.44
#Mann= 5 ,-1 , 0
  3592.7      .1       0  5001.3     .07       0  5007.3      .1       0
  5710.3     .05       0  6291.7      .1       0
Bank Sta=4952.6,5071.4
XS Rating Curve= 0 ,0
Exp/Cntr=0.3,0.1

Type RM Length L Ch R = 1 ,80221   ,78,78,78
BEGIN DESCRIPTION:
UNT003 IN NURI 116.0
END DESCRIPTION:
XS GIS Cut Line= 5
       2300129.7     13345350.03      2299989.09      13345610.4
      2299840.66     13345859.75      2299754.72     13346094.78
       2299338.6     13347153.28
#Sta/Elev= 30
  4312.1  284.62  4446.6  280.12  4455.9  279.92  4489.9  279.04  4495.6  280.59
  4511.8  278.52  4517.5  279.41  4533.7  277.99  4660.9  275.45  4678.3  275.08
  4753.3  273.53  4862.9  273.58  4916.2  272.97  4921.5  270.99  4937.7  271.09
  4977.3  267.27  4998.6  266.84  5001.3  266.34  5004.6  266.84  5007.6  268.19
    5033  271.02  5094.1  272.99  5111.5  273.47  5154.5   274.1  5320.9  273.47
  5504.6  272.78  5751.1  274.29  5971.8  280.48  6070.4  283.04  6285.8  291.71
#Mann= 14 ,-1 , 0
  4312.1      .1       0  4446.6     .08       0  4455.9      .1       0
  4660.9     .08       0  4678.3      .1       0  4862.9     .08       0
  4998.6     .07       0  5004.6     .08       0  5007.6     .05       0
  5111.5      .1       0  5154.5     .08       0  5320.9     .05       0
  5971.8      .1       0  6070.4     .05       0
Bank Sta=4916.2,5094.1
XS Rating Curve= 0 ,0
Exp/Cntr=0.3,0.1

Type RM Length L Ch R = 1 ,80143   ,363,363,363
BEGIN DESCRIPTION:
Mapping XS 053cf15c
END DESCRIPTION:
XS GIS Cut Line= 3
      2300035.99      13345318.7      2299778.16     13345829.15
      2299283.37     13347139.04
#Sta/Elev= 30
    4348  285.46  4498.8  281.48  4521.4  280.69    4570  279.66  4620.9  276.41
  4671.1  277.18  4730.2  275.87  4739.3  275.47  4919.9  271.83  4934.4  271.28
  4974.1  266.48  4989.4  267.38  4991.7  266.38  4994.5  265.88  4997.7  266.38
  5013.6   269.1    5060  271.61  5067.1  272.12  5159.8  274.12  5275.6  273.21
  5291.6  273.94  5373.1  272.55  5477.4  272.58  5786.4     274  6009.5  280.31
    6080  282.27  6200.2  287.42  6253.6  287.72  6292.3   290.3  6320.1  290.48
#Mann= 14 ,-1 , 0
    4348     .08       0  4498.8      .1       0  4521.4     .08       0
  4730.2      .1       0  4739.3     .08       0  4974.1     .05       0
  4991.7     .03       0  4997.7     .05       0    5060     .08       0
  5275.6     .05       0  5373.1     .08       0  5477.4     .05       0
  6009.5      .1       0    6080     .05       0
Bank Sta=4919.9,5067.1
XS Rating Curve= 0 ,0
Exp/Cntr=0.3,0.1

Type RM Length L Ch R = 1 ,79780   ,412,412,412
BEGIN DESCRIPTION:
UNT003 IN NURI 115.0
END DESCRIPTION:
XS GIS Cut Line= 3
      2299637.71     13345396.87      2299437.72     13345746.85
      2299037.72     13346946.85
#Sta/Elev= 30
  4607.8  284.27  4641.9  282.71  4696.3  280.54  4739.5  280.12  4761.1  278.64
  4776.9  278.99  4863.3  276.56  4930.3  273.09  4953.3   270.6  4959.8  267.97
  4994.2   262.1    4997   261.6  5000.2   262.1  5013.5  262.47  5042.5  268.85
  5063.6  270.72  5190.1  272.22  5274.4  270.96  5379.8  271.88  5569.6   271.2
  5601.2  272.81  5611.7  271.83  5653.9  271.26  5727.7  271.23  5864.7  275.35
  5949.2  279.54  6001.7  281.08  6012.3  282.27  6138.8  287.51  6275.8     292
#Mann= 5 ,-1 , 0
  4607.8      .1       0  4641.9     .05       0  4994.2    .035       0
  5000.2     .05       0  5949.2      .1       0
Bank Sta=4953.3,5063.6
XS Rating Curve= 0 ,0
Exp/Cntr=0.3,0.1

Type RM Length L Ch R = 1 ,79368   ,471,471,471
BEGIN DESCRIPTION:
UNT003 IN NURI 114.0
END DESCRIPTION:
XS GIS Cut Line= 4
      2299549.01     13345186.56      2299127.11     13345418.35
      2298942.22     13345931.37      2298955.24     13346840.18
#Sta/Elev= 30
    4340  284.87  4392.7  283.47    4524  276.81  4642.8  272.38  4664.6   273.7
  4680.7  271.96  4752.2  270.34  4936.7  271.29  4952.5  269.26  4977.9  263.64
  4997.5  260.94  5000.2  260.44  5003.5  260.94  5032.4  265.94  5044.6  269.88
  5064.3  271.59  5085.5  270.33    5162  271.06  5266.2  269.79  5462.2  270.91
  5522.2  269.93  5732.2  270.34  5802.2  271.62  5964.8  278.36  5992.3  279.27
  6012.3  278.09  6039.8  279.59  6112.3  284.21  6159.7  285.68  6275.6  289.18
#Mann= 6 ,-1 , 0
    4340     .05       0  4997.5     .03       0  5003.5     .05       0
  5964.8     .08       0  6039.8     .05       0  6159.7      .1       0
Bank Sta=4952.5,5044.6
XS Rating Curve= 0 ,0
Exp/Cntr=0.3,0.1

Type RM Length L Ch R = 1 ,78897   ,347,347,347
BEGIN DESCRIPTION:
UNT003 IN NURI 113.0
END DESCRIPTION:
XS GIS Cut Line= 3
      2299737.74     13344796.84      2298637.72     13345396.85
      2297537.74     13345896.85
#Sta/Elev= 30
  3746.9  295.32  3872.2  292.07    3924  289.24  3945.8  289.74  4365.4  273.23
  4387.2  275.02  4425.2  272.12  4653.9  268.48  4794.9  271.13  4888.4  270.86
  4942.5  268.56  4988.8  259.94  4991.6  259.44  4994.8  259.94  5031.8  263.96
  5037.3  266.24  5088.9   268.7  5164.7  269.77  5337.9  267.84  5399.8  264.43
  5474.5  263.14  5515.1  267.08  5594.8  270.94    5626  273.69  5641.4  273.09
  5733.7  277.39  5756.8  279.92  5813.5  282.85  5937.6  288.99  6208.2  298.52
#Mann= 8 ,-1 , 0
  3746.9     .05       0  4988.8     .03       0  4994.8     .05       0
  5337.9      .1       0  5594.8     .05       0  5756.8      .1       0
  5813.5     .05       0  5937.6      .1       0
#XS Ineff= 1 ,-1
 5174.88 5585.61  269.67
Permanent Ineff=
       F
Bank Sta=4942.5,5088.9
XS Rating Curve= 0 ,0
Exp/Cntr=0.3,0.1

Type RM Length L Ch R = 1 ,78550   ,722,722,722
BEGIN DESCRIPTION:
UNT003 IN NURI 112.0
END DESCRIPTION:
XS GIS Cut Line= 4
       2299696.1     13344665.94      2298984.28     13344888.17
      2298189.14     13345349.97      2297393.98     13345603.45
#Sta/Elev= 30
  3477.8  294.49  3667.7  289.63  3938.1  278.78  4094.2  277.27  4219.1  273.34
  4249.6  274.87  4484.7  268.21    4578  266.81  4752.9   270.1  4878.6  268.27
  4913.5  268.05  4972.3  260.39  5000.7  259.02  5003.5  258.52  5006.7  259.02
  5062.5  268.17  5089.8  269.35  5144.4   266.8  5218.8  265.35  5246.1  261.79
  5267.5  262.37  5291.4  266.09  5440.5  274.55  5469.9  277.67  5501.4  277.16
  5752.8  291.26  5856.8  294.93  5951.8  298.16    5959  298.12  5977.6  298.45
#Mann= 12 ,-1 , 0
  3477.8     .05       0  4878.6      .1       0  5000.7     .07       0
  5006.7      .1       0  5144.4     .05       0  5218.8      .1       0
  5267.5     .05       0  5440.5      .1       0  5752.8     .05       0
  5856.8      .1       0  5951.8     .05       0    5959      .1       0
#XS Ineff= 1 ,-1
 5089.96 5361.69  269.36
Permanent Ineff=
       F
Bank Sta=4913.5,5062.5
XS Rating Curve= 0 ,0
Exp/Cntr=0.3,0.1

Type RM Length L Ch R = 1 ,77828   ,519,519,519
BEGIN DESCRIPTION:
UNT003 IN NURI 110.0
END DESCRIPTION:
XS GIS Cut Line= 3
      2299593.28     13344489.19      2298742.32     13344466.19
      2296902.98     13345201.93
#Sta/Elev= 30
  3081.4  288.24  3617.2  276.28  3897.3  275.48  3959.2  273.66  3980.7  275.37
  4058.6  271.47  4322.4  265.92  4824.5  266.95  4928.5  266.36    4974  262.16
  4995.3  257.94    4998  257.44  5001.3  257.94  5031.2  261.29  5081.7  265.61
    5351  277.09  5380.8  280.37  5399.5  279.75  5562.6  289.96  5660.9  296.71
  5800.7  301.69  5811.7  304.61  5830.3  305.05  5835.7  299.02  5865.5   296.6
  5876.3  297.13  5884.1  303.33  5889.5  300.95  5897.8   306.2  5913.7  304.66
#Mann= 6 ,-1 , 0
  3081.4     .05       0  4824.5      .1       0  4995.3     .07       0
  5001.3      .1       0  5031.2     .05       0  5562.6      .1       0
Bank Sta=4928.5,5081.7
XS Rating Curve= 0 ,0
Exp/Cntr=0.3,0.1

Type RM Length L Ch R = 1 ,77309   ,936,936,936
BEGIN DESCRIPTION:
UNT003 IN NURI 109.0
END DESCRIPTION:
XS GIS Cut Line= 3
      2299156.29     13343776.22      2298454.83      13344040.7
      2296775.86     13344684.69
#Sta/Elev= 30
  3289.7   282.3  3437.8  278.58  3450.6  279.47  3598.1  273.77  3608.8  275.38
  3676.2  272.59  3801.2  272.77  3854.6  274.88  3871.6  273.12  3918.7  274.82
  4017.3   274.6    4321  264.15  4689.9   265.9  4902.3  264.18  4933.4  264.83
  4957.4  262.96  4997.2  257.06  4999.9  256.56  5003.2  257.06  5038.6  260.57
  5108.2  264.37    5327  275.36  5460.7  279.15  5630.5  286.72  5685.2  287.56
  5696.4  289.41  5728.5  289.71  5750.6  292.17    5830  295.73  5837.6  294.98
#Mann= 5 ,-1 , 0
  3289.7     .05       0  4902.3      .1       0  4997.2     .07       0
  5003.2      .1       0  5038.6     .05       0
Bank Sta=4933.4,5108.2
XS Rating Curve= 0 ,0
Exp/Cntr=0.3,0.1

Type RM Length L Ch R = 1 ,76373   ,461,461,461
BEGIN DESCRIPTION:
UNT003 IN NURI 108.0
END DESCRIPTION:
XS GIS Cut Line= 3
      2298587.69     13342846.87      2297187.72     13343546.85
      2296637.71     13343946.86
#Sta/Elev= 30
  3464.8  290.42  3621.3  284.13    3652  284.05  3763.8  278.51  3830.9  277.22
  3867.3  274.05    3898  275.36  3922.8   273.3  3929.1  272.97  4263.5  262.49
  4708.6  263.04  4820.4  259.66  4932.2  262.15  4971.3  259.11  4985.3  255.41
  4996.3  254.68    4999  254.18  5002.3  254.68    5016  255.88  5027.2  258.64
  5108.5  262.18  5351.5  271.63  5466.3  274.94  5487.5  274.44  5545.9  277.72
  5574.1  277.02  5631.6  280.34  5652.5   279.9  5702.7  283.29  5710.1  282.43
#Mann= 6 ,-1 , 0
  3464.8      .1       0  3922.8     .05       0  3929.1      .1       0
  4263.5     .05       0  4996.3     .03       0  5002.3     .05       0
Bank Sta=4932.2,5108.5
XS Rating Curve= 0 ,0
Exp/Cntr=0.3,0.1

Type RM Length L Ch R = 1 ,75912   ,630,630,630
BEGIN DESCRIPTION:
UNT003 IN NURI 107.0
END DESCRIPTION:
XS GIS Cut Line= 3
       2298500.8     13342511.25      2297661.35     13342683.74
      2296362.31     13343557.43
#Sta/Elev= 30
  3352.8  286.02  3539.7   280.8  3554.8  281.59  3570.3  279.54  3580.5  281.16
  3631.6  280.58  3672.4  277.22  3733.7  277.69  3866.4   273.2  4142.1  269.26
  4264.3   266.9  4480.3  259.23  4756.2   260.4  4891.2  259.21  4937.3  260.54
  4978.2   259.1  5005.1  252.91  5007.9  252.41  5011.1  252.91  5044.1  258.62
  5056.6  258.54  5245.1  267.65  5281.1  267.19  5491.1  275.36  5527.1  274.89
    5563  277.67  5584.1  276.81  5648.3  280.27  5677.1  279.56  5775.3  283.18
#Mann= 6 ,-1 , 0
  3352.8      .1       0  4142.1     .05       0  4937.3      .1       0
  5005.1     .07       0  5011.1      .1       0  5056.6     .05       0
Bank Sta=4978.2,5044.1
XS Rating Curve= 0 ,0
Exp/Cntr=0.3,0.1

Type RM Length L Ch R = 1 ,75282   ,468,468,468
BEGIN DESCRIPTION:
UNT003 IN NURI 106.0
END DESCRIPTION:
XS GIS Cut Line= 4
      2298397.33     13341338.28      2297569.35     13342143.25
      2296350.39     13342752.74      2295971.78     13342787.16
#Sta/Elev= 30
  2940.7  289.47    3187  281.92    3394  278.36  3422.8  277.61  3523.7  274.93
  3879.9  266.12  4427.4  257.77  4849.3  257.59  4935.8  259.54  4964.1  258.03
  4999.9  252.36  5002.7  251.86  5005.9  252.36  5031.2  257.15  5049.3  256.27
  5092.4  258.17  5120.6  257.32  5159.4  260.04  5181.8  258.53  5254.8  263.78
  5293.6  262.91  5366.6   268.2  5405.4  266.57  5491.1  271.47  5521.3  270.61
  5601.6  275.25  5631.7  274.76    5702  279.19  5722.1  278.07  5838.5  283.06
#Mann= 8 ,-1 , 0
  2940.7      .1       0    3394     .05       0  3422.8      .1       0
  3523.7     .05       0  4849.3      .1       0  4999.9     .07       0
  5005.9      .1       0  5049.3     .05       0
Bank Sta=4964.1,5092.4
XS Rating Curve= 0 ,0
Exp/Cntr=0.3,0.1

Type RM Length L Ch R = 1 ,74814   ,514,514,514
BEGIN DESCRIPTION:
UNT003 IN NURI 105.0
END DESCRIPTION:
XS GIS Cut Line= 3
      2298087.72     13340546.86      2296537.72     13342146.85
      2296137.69     13342446.88
#Sta/Elev= 30
  2780.8  298.84  2901.1  294.83  2922.2  296.06    3145  287.72  3632.5  271.96
  3650.7  271.59  4053.7  260.94  4301.2  257.48  4768.1  255.98  4859.9  258.75
  4973.1  256.86  4998.4  249.31  5001.1  248.81  5004.4  249.31    5005  252.28
    5030  256.02  5036.6  257.05    5072  254.46  5118.8  257.07  5158.5  260.33
  5180.3  259.09  5215.8  263.95  5251.2  263.68  5286.6  268.23  5308.5  267.02
  5351.2  271.56    5372  270.55  5436.6  275.47  5458.5  274.45  5508.5  277.34
#Mann= 8 ,-1 , 0
  2780.8      .1       0    3145     .05       0  3632.5      .1       0
  3650.7     .05       0  4998.4    .035       0  5004.4     .05       0
    5030      .1       0  5118.8     .05       0
Bank Sta=4973.1,5036.6
XS Rating Curve= 0 ,0
Exp/Cntr=0.3,0.1

Type RM Length L Ch R = 1 ,74300   ,497,497,497
BEGIN DESCRIPTION:
UNT003 IN NURI 104.0
END DESCRIPTION:
XS GIS Cut Line= 3
      2297637.72     13340596.86      2296237.72     13341746.85
      2295787.69     13342196.89
#Sta/Elev= 30
  3189.9  288.98  3310.4  283.89  3332.2  285.06    3446  279.67  3557.2  274.86
    3837  263.72  4134.6  256.83  4405.4   254.6  4710.3  256.03  4809.4   254.2
  4937.1  256.21  4980.1  253.86  4994.5  251.52  4995.4  247.85  4998.2  247.35
  5001.4  247.85  5029.9  253.52  5058.2  255.28  5086.5  254.08  5143.1  255.78
  5213.8  260.68  5242.1  259.94  5298.6  264.56  5341.1  264.27  5397.6  268.31
  5425.9  267.37  5468.4   271.6  5482.5  270.51  5623.9  278.88  5638.1  278.05
#Mann= 5 ,-1 , 0
  3189.9     .05       0    3446      .1       0  3557.2     .05       0
  4995.4    .035       0  5001.4     .05       0
Bank Sta=4937.1,5058.2
XS Rating Curve= 0 ,0
Exp/Cntr=0.3,0.1

Type RM Length L Ch R = 1 ,73803   ,549,549,549
BEGIN DESCRIPTION:
UNT003 IN NURI 103.0
END DESCRIPTION:
XS GIS Cut Line= 3
      2297587.74     13340546.85      2296187.72     13341246.85
      2295537.69     13341846.88
#Sta/Elev= 30
  3397.7  287.84  3478.8  284.44  3501.1  285.27    3678  277.12  3741.8  274.12
  4121.6  259.44  4202.7  257.83  4546.5  253.71    4751  254.21  4883.4  254.23
  4918.2  253.14  4926.6  251.45  4940.6  252.18    4949  248.62  4954.6  250.65
  4966.4  250.68  4970.1  247.49  4981.2  247.41    4984  246.91  4987.2  247.41
  5005.2   247.8  5012.6  251.67  5040.9  253.21  5224.7  255.04  5295.5  257.48
  5316.8  256.02  5507.6  264.36  5529.2  263.03  5568.4  265.67  5847.6  277.03
#Mann= 8 ,-1 , 0
  3397.7     .05       0    3678      .1       0  3741.8     .05       0
    4751      .1       0  4883.4     .05       0  4981.2    .035       0
  4987.2     .05       0  5568.4      .1       0
Bank Sta=4918.2,5040.9
XS Rating Curve= 0 ,0
Exp/Cntr=0.3,0.1

Type RM Length L Ch R = 1 ,73254   ,571,571,571
BEGIN DESCRIPTION:
UNT003 IN NURI 102.0
END DESCRIPTION:
XS GIS Cut Line= 3
      2296807.64     13340251.91      2295904.42     13340915.94
      2295442.64     13341787.41
#Sta/Elev= 30
  4159.8  272.89  4357.2  266.64  4528.5  258.94  4670.5  253.74  4720.6  252.43
  4815.9  251.92  4956.7     253  4971.4  252.13  4997.7     246  5000.4   245.5
  5003.7     246  5006.9  247.45  5028.5  251.11  5050.8  250.87  5086.3  252.96
  5136.2  253.09  5251.4  252.49  5383.7  256.06  5544.3  256.55  5582.6  258.04
  5610.3  256.59  5670.6  259.17    5678   260.3  5692.6  260.32    5709  258.93
  5736.6  260.61  5808.9  262.27  5938.3  267.62  6017.5  269.12  6267.1  276.39
#Mann= 6 ,-1 , 0
  4159.8     .05       0  4815.9      .1       0  4997.7     .07       0
  5003.7      .1       0  5136.2     .05       0  5808.9      .1       0
Bank Sta=4956.7,5086.3
XS Rating Curve= 0 ,0
Exp/Cntr=0.3,0.1

Type RM Length L Ch R = 1 ,72683   ,416,416,416
BEGIN DESCRIPTION:
UNT003 IN NURI 101.0
END DESCRIPTION:
XS GIS Cut Line= 3
      2296737.67     13340196.86      2295787.72     13340296.85
      2294187.73     13340796.85
#Sta/Elev= 30
  4054.1  272.27  4384.6  261.45  4496.5  256.17  4728.1  249.93  4771.7  251.42
  4788.1  251.12  4808.2  248.55  4828.3  249.05  4848.4  251.42  4928.9  251.41
  4938.9  250.05  4969.1  249.79  4996.2  244.93    4999  244.43  5002.2  244.93
  5030.8  247.22  5051.2  247.12    5058  248.92  5063.3  248.46  5090.5  251.72
  5230.9  250.42  5386.5  251.04  5805.5  262.09  5973.2  263.58    6057  266.34
  6166.5  267.35  6193.2  269.05  6423.7  275.34    6464  277.38  6685.6  283.09
#Mann= 4 ,-1 , 0
  4054.1     .05       0  4728.1      .1       0  4996.2     .07       0
  5002.2      .1       0
Bank Sta=4928.9,5090.5
XS Rating Curve= 0 ,0
Exp/Cntr=0.3,0.1

Type RM Length L Ch R = 1 ,72267   ,484,484,484
BEGIN DESCRIPTION:
UNT003 IN NURI 100.0
END DESCRIPTION:
XS GIS Cut Line= 3
      2296545.89     13339935.32       2296016.9     13339762.82
      2294131.85     13340555.92
#Sta/Elev= 30
  3959.6  268.23  4189.1  263.12  4259.3  260.32  4487.9  257.68  4558.5  255.45
  4741.6  252.01  4753.8  250.16    4808   248.8  4947.8  250.82  4959.9  248.27
  4970.8  248.11  4982.4  245.69  4992.5  245.12  4997.7  243.35  5000.4  242.85
  5003.7  243.35  5024.4   247.5  5090.1  250.72  5336.4  248.72  5372.2   250.8
  5578.3   256.6  5784.5  261.11  5801.8   260.3  6037.2   264.3  6190.5  269.23
  6207.6   271.1  6261.7  271.72  6372.9  276.33  6396.7  275.88  6561.1  282.19
#Mann= 4 ,-1 , 0
  3959.6     .05       0  4558.5      .1       0  4997.7     .07       0
  5003.7      .1       0
Bank Sta=4947.8,5090.1
XS Rating Curve= 0 ,0
Exp/Cntr=0.3,0.1

Type RM Length L Ch R = 1 ,71783   ,664,664,664
BEGIN DESCRIPTION:
UNT003 IN NURI 99.0
END DESCRIPTION:
XS GIS Cut Line= 3
      2296200.89     13339521.33      2295694.91     13339371.83
      2293832.32     13340337.62
#Sta/Elev= 30
  3956.9  264.59  4198.5  264.98  4408.6  261.55    4560  256.94  4592.5  255.96
  4640.7  255.49  4819.3  246.86  4954.4  247.32    4989   245.5  4996.5  241.98
  4999.2  241.48  5002.5  241.98  5004.7     242  5033.3  247.84  5110.5  248.63
  5200.3   246.6  5236.4  247.28  5376.5  249.46    5623  254.14  5799.3  257.99
  5962.2  264.04  5990.8  262.93  6168.5  267.91    6285  272.33  6421.2  274.54
  6526.2  277.57  6531.9  279.41  6564.8  279.41  6570.5  280.92  6582.6  280.03
#Mann= 12 ,-1 , 0
  3956.9     .05       0    4560      .1       0  4592.5     .16       0
  4996.5     .07       0  5002.5     .16       0  5004.7      .1       0
  5200.3     .16       0  5236.4      .1       0  5376.5     .16       0
    5623      .1       0  6168.5     .16       0    6285      .1       0
Bank Sta=4954.4,5033.3
XS Rating Curve= 0 ,0
Exp/Cntr=0.3,0.1

Type RM Length L Ch R = 1 ,71119   ,573,573,573
BEGIN DESCRIPTION:
UNT003 IN NURI 98.0
END DESCRIPTION:
XS GIS Cut Line= 4
      2296706.55     13338919.42      2295439.14     13338961.08
      2294886.55     13339143.87      2293787.71     13339946.86
#Sta/Elev= 30
  3408.9  267.61  3657.9  265.78  4028.1  256.84  4258.2  253.49  4468.3  253.39
  4675.2  256.71  4775.7  254.34  4854.8  252.31  4961.8   246.6  4993.5  241.27
  4995.8  239.69  4998.6  239.19  5001.8  239.69  5025.3  242.17  5036.6  245.34
  5068.2  245.96  5110.3   245.1  5278.2  246.89  5374.7  246.62  5454.3  243.78
    5516  246.88  5839.7  250.36  5989.5  255.23  6062.6  259.87  6126.1  261.86
  6384.7  272.91  6462.1  277.59  6551.9  280.36  6583.3  282.52    6620  281.65
#Mann= 9 ,-1 , 0
  3408.9     .05       0  4775.7      .1       0  4854.8     .16       0
  4995.8     .07       0  5001.8     .16       0  5278.2      .1       0
    5516     .16       0  6126.1      .1       0  6551.9     .05       0
Bank Sta=4961.8,5068.2
XS Rating Curve= 0 ,0
Exp/Cntr=0.3,0.1

Type RM Length L Ch R = 1 ,70546   ,563,563,563
BEGIN DESCRIPTION:
UNT003 IN NURI 97.0
END DESCRIPTION:
XS GIS Cut Line= 4
      2296689.96      13338873.4      2295101.46     13338508.83
      2294481.01     13338700.21      2293547.61     13339324.82
#Sta/Elev= 30
  3063.7  267.46  3230.2  266.47  3744.7  255.59  4040.7  253.34    4133  250.99
  4225.4  253.38  4399.8  254.87  4668.7  250.71  4777.3  249.06  4827.9  248.09
  4885.8   246.4  4917.2   243.9    4975   244.2  4997.9  238.51  5000.6  238.01
  5003.9  238.51  5021.8  243.95  5032.3   244.5  5126.5  243.14  5189.3  244.35
  5279.4  243.14  5332.8  243.88  5358.3  244.95  5484.9  245.03  5528.1  245.61
  5599.8  246.71  5752.4  249.44    5885   254.5  6048.8  257.37  6465.9  271.98
#Mann= 12 ,-1 , 0
  3063.7     .05       0  4668.7      .1       0  4777.3     .16       0
  4827.9      .1       0  4997.9     .07       0  5003.9      .1       0
  5332.8     .05       0  5484.9      .1       0  5528.1     .05       0
  5599.8      .1       0  5752.4     .05       0    5885      .1       0
Bank Sta=4975,5032.3
XS Rating Curve= 0 ,0
Exp/Cntr=0.3,0.1

Type RM Length L Ch R = 1 ,69983   ,811,811,811
BEGIN DESCRIPTION:
UNT003 IN NURI 96.0
END DESCRIPTION:
XS GIS Cut Line= 3
      2295999.01     13337363.01      2295075.42      13337974.1
      2293384.42     13338404.67
#Sta/Elev= 30
  3512.9  257.35  3532.8  256.64  3679.6  250.62  3885.8  243.34    3985  244.22
  3994.1  243.83  4006.1  240.31  4021.1   243.7  4042.2  244.26    4066  243.18
  4129.5  244.48  4186.6  242.88  4309.4  243.01  4596.6  244.65  4734.7  244.15
  4857.4  241.47  4958.5  242.86  4980.1  241.04  4996.8  237.08  4999.5  236.58
  5002.8  237.08  5030.7  243.33  5051.4  244.87  5123.6  246.02  5155.5  244.52
  5397.5  242.87  5595.8  243.23  5856.3  247.09  6012.4  254.32  6365.3  267.63
#Mann= 11 ,-1 , 0
  3512.9     .08       0  3532.8     .05       0  3679.6      .1       0
  4309.4     .05       0  4596.6      .1       0  4996.8     .07       0
  5002.8      .1       0  5155.5     .05       0  5397.5      .1       0
  5595.8     .05       0  6012.4      .1       0
#XS Ineff= 1 ,-1
 3973.44 4130.47  244.56
Permanent Ineff=
       F
Bank Sta=4958.5,5030.7
XS Rating Curve= 0 ,0
Exp/Cntr=0.3,0.1

Type RM Length L Ch R = 1 ,69172   ,115,115,115
BEGIN DESCRIPTION:
UNT003 IN NURI 95.0
END DESCRIPTION:
XS GIS Cut Line= 3
      2295880.95     13337293.55       2294540.7     13337307.44
      2293964.29      13337425.5
#Sta/Elev= 30
    3980  256.33  4072.6  254.15  4533.3  242.44  4693.3  242.55  4753.3  241.99
  4793.3  240.69  4863.3  240.33  4913.3  241.53  4943.3  241.28  4953.3  240.55
  4963.3  238.35  4973.3  238.96  5000.3  237.83    5003  237.33  5006.3  237.83
  5013.3  239.66  5023.3  240.09  5043.3  238.65  5083.3  240.39  5143.3  240.36
  5183.3  242.67  5213.3  242.98  5253.3  244.68  5283.3  246.64  5527.5  250.28
    5701  254.32  5731.7   256.6  5792.1  257.47  5813.3  258.09  5908.7  257.15
#Mann= 5 ,-1 , 0
    3980     .08       0  4072.6     .05       0  5000.3     .04       0
  5006.3     .05       0  5792.1      .1       0
Bank Sta=4943.3,5023.3
XS Rating Curve= 0 ,0
Exp/Cntr=0.3,0.1

Type RM Length L Ch R = 1 ,69057   ,453,453,453
BEGIN DESCRIPTION:
UNT003 IN NURI 94.0
END DESCRIPTION:
XS GIS Cut Line= 3
      2295964.31     13337234.52      2294530.28     13337175.49
      2293892.09     13337255.27
#Sta/Elev= 30
  3892.2  260.31  3928.8  258.23  3955.4   257.7  3960.4  258.78  4038.9  255.63
    4159  253.18  4419.2  244.76  4729.5  240.12  4959.7  240.16  4979.7  239.61
  4996.7   236.7  4999.5   236.2  5002.7   236.7  5019.7  236.82  5049.8  239.64
  5069.8  240.32  5168.8   238.9  5173.8  237.99  5244.6  240.37    5290  241.39
  5342.9  245.86  5382.1  247.48  5442.3  247.63  5618.9  249.66    5624  251.12
  5652.5  250.75  5704.6  252.55  5780.2  252.97  5865.8  255.18  5970.6  255.57
#Mann= 6 ,-1 , 0
  3892.2      .1       0  4996.7     .07       0  5002.7      .1       0
  5244.6     .05       0  5342.9      .1       0  5442.3     .05       0
Bank Sta=4959.7,5069.8
XS Rating Curve= 0 ,0
Exp/Cntr=0.3,0.1

Type RM Length L Ch R = 1 ,68604   ,436,436,436
BEGIN DESCRIPTION:
Mapping XS 0b025cd8
END DESCRIPTION:
XS GIS Cut Line= 3
      2295891.43     13336637.29      2294308.06     13336821.33
      2293899.69     13337233.16
#Sta/Elev= 30
  3819.5  272.83  3863.8  270.26  3873.6  270.89  3942.3  265.59  3994.4  264.54
  4044.7  260.43  4095.1  259.04  4114.5  259.86  4135.3  257.05  4346.7  248.66
  4427.3   247.2  4463.9  244.56  4719.2  239.13  4900.3  237.63  4970.9  238.83
  4985.5  238.42  4998.1  234.45  5000.9  233.95  5004.1  234.45  5021.2  239.38
  5246.1  240.35  5495.4  246.77  5530.8     246  5636.9  247.43  5658.1     249
  5686.4  248.39    5743  249.82  5778.3  251.95  5827.8  251.54  5993.5  254.46
#Mann= 5 ,-1 , 0
  3819.5     .05       0  4900.3      .1       0  4998.1     .07       0
  5004.1      .1       0  5246.1     .05       0
Bank Sta=4970.9,5021.2
XS Rating Curve= 0 ,0
Exp/Cntr=0.3,0.1

Type RM Length L Ch R = 1 ,68168   ,803,803,803
BEGIN DESCRIPTION:
Mapping XS c474fe4c
END DESCRIPTION:
XS GIS Cut Line= 3
      2295502.49     13336015.78      2294342.78     13336481.05
      2293832.57      13337248.1
#Sta/Elev= 30
  4007.2  266.52  4055.6   264.1  4074.4  264.38  4163.2  259.21    4182   259.6
  4217.1  256.64  4303.3  252.82  4319.2   253.2  4402.6  248.58    4451  246.73
  4464.9  247.09  4510.2   244.5  4604.9  241.16  4809.7  237.29  4875.4  237.54
  4940.5  238.25  4982.1  237.63  4994.3  236.34  5000.6  233.85  5003.4  233.35
  5006.6  233.85  5013.1   234.1  5025.2  238.55  5100.9  237.82  5350.5  240.85
  5581.9  248.82  5891.5   250.5  6035.8  253.91  6056.9  253.07    6178  254.49
#Mann= 5 ,-1 , 0
  4007.2     .05       0  4875.4      .1       0  5000.6     .07       0
  5006.6      .1       0  5100.9     .05       0
Bank Sta=4982.1,5025.2
XS Rating Curve= 0 ,0
Exp/Cntr=0.3,0.1

Type RM Length L Ch R = 1 ,67365   ,615,615,615
BEGIN DESCRIPTION:
UNT003 IN NURI 93.0
END DESCRIPTION:
XS GIS Cut Line= 3
      2295134.41     13335494.95       2294228.2     13335731.05
       2293752.8     13337282.17
#Sta/Elev= 30
    4156  261.95  4255.9  259.85  4337.7  255.36  4423.9  252.84  4472.9  249.02
  4524.6  247.95  4540.2  246.32  4555.6  247.37  4627.9  243.94  4915.2  235.96
    4969  236.39  4989.6   232.9  5007.3  232.59    5010  232.09  5013.3  232.59
  5021.1  235.38  5041.3  236.46  5132.9   235.2  5347.2  237.67  5464.6  236.16
  5695.6  241.87  5755.9  242.13  5799.3  244.73  5831.9  244.38  5897.4  247.12
  5977.1  247.26  6018.9  249.26  6033.6  248.24  6290.9  249.02  6714.8  254.52
#Mann= 5 ,-1 , 0
    4156     .05       0  4915.2      .1       0  5007.3     .07       0
  5013.3      .1       0  5132.9     .05       0
Bank Sta=4969,5041.3
XS Rating Curve= 0 ,0
Exp/Cntr=0.3,0.1

Type RM Length L Ch R = 1 ,66750   ,582,582,582
BEGIN DESCRIPTION:
UNT003 IN NURI 92.0
END DESCRIPTION:
XS GIS Cut Line= 3
      2293908.75     13334781.43      2293736.88     13335828.27
      2293663.96     13337208.49
#Sta/Elev= 30
  4349.9  261.75  4511.5  256.01  4537.8  253.82  4608.7  251.54  4618.9   249.9
    4634  250.12  4695.3  245.69  4720.2  245.68  4756.6   242.5  4840.8  239.42
  4940.4  233.99  4963.4  234.81  4973.6  234.59  4998.6   229.5  5001.4     229
  5004.6   229.5  5006.7  232.14  5014.1  234.55  5024.2   235.6  5095.2  233.13
  5196.5  235.71  5439.4  235.67  5549.5  237.12  6070.3  249.08  6240.5  249.12
  6350.6  247.38  6436.6  248.87  6470.8  247.97  6651.1  251.72  6792.9  252.19
#Mann= 5 ,-1 , 0
  4349.9     .05       0  4840.8      .1       0  4998.6     .07       0
  5004.6      .1       0  5095.2     .05       0
Bank Sta=4963.4,5024.2
XS Rating Curve= 0 ,0
Exp/Cntr=0.3,0.1

Type RM Length L Ch R = 1 ,66168   ,528,528,528
BEGIN DESCRIPTION:
UNT003 IN NURI 91.0
END DESCRIPTION:
XS GIS Cut Line= 4
       2293577.5     13334747.69      2293327.93     13334953.86
       2292915.6     13336592.32      2292926.44     13336852.33
#Sta/Elev= 30
  4279.3   259.8  4356.8  257.42  4438.9  252.63  4894.8   233.6  4925.8  233.11
  4977.3  234.31  4987.6  232.77  4995.1  226.84  4997.9  226.34  5001.1  226.84
  5028.9  234.09  5101.1  232.47  5157.4  233.01  5173.3  234.62  5214.5  233.63
  5269.2  234.54  5400.6  235.57  5552.9  237.52  5808.1  239.13  5884.8   239.7
  5915.7  241.57  5946.6  240.42  6020.8  242.66    6031   244.1  6061.9  243.06
  6152.9  246.89    6180  246.16  6235.4  247.59  6363.8  248.16  6552.8  248.08
#Mann= 10 ,-1 , 0
  4279.3     .05       0  4438.9      .1       0  4995.1     .07       0
  5001.1      .1       0  5269.2     .05       0  5400.6      .1       0
  5552.9     .05       0  5808.1      .1       0    6031     .05       0
  6363.8      .1       0
Bank Sta=4977.3,5028.9
XS Rating Curve= 0 ,0
Exp/Cntr=0.3,0.1

Type RM Length L Ch R = 1 ,65640   ,430,430,430
BEGIN DESCRIPTION:
UNT003 IN NURI 90.0
END DESCRIPTION:
XS GIS Cut Line= 3
      2292837.72     13334496.86      2292676.96      13335511.2
      2292188.39     13336430.77
#Sta/Elev= 30
  4180.2  258.02  4301.7  254.23  4343.6  251.67  4392.8  250.35  4777.6   233.5
  4852.2  232.59  4959.8  233.75  4969.9  232.94  4976.9  230.47  4981.9  231.38
  4990.2  230.67  5000.3  226.12  5007.4  225.96  5010.2  225.46  5013.4  225.96
  5020.6  231.59  5030.7  232.43  5071.2  232.23  5091.4  233.44  5440.1  235.07
  5667.4   235.9  5794.2  236.11  5898.5  237.69  6040.2  242.24  6090.6  242.66
  6128.9  244.46  6150.9  244.07  6156.6  245.14  6168.3  244.42  6248.5  245.71
#Mann= 6 ,-1 , 0
  4180.2      .1       0  5007.4     .07       0  5013.4      .1       0
  5440.1     .16       0  5667.4      .1       0  6168.3     .05       0
Bank Sta=4959.8,5091.4
XS Rating Curve= 0 ,0
Exp/Cntr=0.3,0.1

Type RM Length L Ch R = 1 ,65210   ,508,508,508
BEGIN DESCRIPTION:
UNT003 IN NURI 89.0
END DESCRIPTION:
XS GIS Cut Line= 3
      2292787.72     13334446.85      2292287.72     13335246.85
      2290987.72     13336796.86
#Sta/Elev= 30
  4054.2   258.8  4207.5   253.7  4685.7  233.51  4764.7   231.6  4962.2  231.63
  4974.6  230.91  4989.9  226.79  4991.7  224.59  4994.4  224.09  4997.7  224.59
  5000.9  224.59  5004.8  229.07  5019.1  232.31  5082.8  233.24  5238.9  232.53
  5267.5   229.6  5302.7  232.75  5359.9  233.35  5707.3  234.67  5941.5  237.75
  6232.9  239.65  6431.9  244.62    6588  249.97  6594.5  248.46  6602.3  250.16
  6651.8  250.37  6812.7   255.4  6836.5  256.76  6858.1  256.13  7020.6  259.01
#Mann= 5 ,-1 , 0
  4054.2      .1       0  4991.7     .07       0  4997.7      .1       0
  6812.7     .08       0  6858.1      .1       0
Bank Sta=4962.2,5019.1
XS Rating Curve= 0 ,0
Exp/Cntr=0.3,0.1

Type RM Length L Ch R = 1 ,64702   ,631,631,631
BEGIN DESCRIPTION:
UNT003 IN NURI 88.0
END DESCRIPTION:
XS GIS Cut Line= 3
      2292537.69     13334446.88      2291787.72     13335096.85
      2291087.71     13336346.87
#Sta/Elev= 30
  4037.3  253.86    4165  248.89  4179.3  246.92  4200.1  247.18  4355.9  240.91
  4398.6  238.01  4725.4  231.64  4752.9   230.7  4767.1   228.6  4973.2  231.18
  4987.5  229.64  4994.1   223.3  4998.7  223.19  5001.5  222.69  5004.7  223.19
  5008.4  225.26    5016  226.17  5022.6  229.43  5032.6  228.82  5043.4  231.69
  5075.4   233.1  5162.1  230.04  5405.3  232.23  5763.3     240  6095.6  242.19
  6345.9  249.37  6405.1   249.5    6427   251.9  6439.5  250.74  6462.4   251.8
#Mann= 3 ,-1 , 0
  4037.3      .1       0  4998.7     .07       0  5004.7      .1       0
Bank Sta=4973.2,5043.4
XS Rating Curve= 0 ,0
Exp/Cntr=0.3,0.1

Type RM Length L Ch R = 1 ,64071   ,714,714,714
BEGIN DESCRIPTION:
Mapping XS b42150c1
END DESCRIPTION:
XS GIS Cut Line= 3
      2292502.46     13334067.88      2291080.63     13334791.81
      2291075.42     13336307.48
#Sta/Elev= 30
  3749.3   255.8  4064.9  244.32  4181.7  237.85  4409.8  232.08  4428.5  232.01
  4732.2  231.38  4854.3  227.51    4860  224.06  4876.6   223.7    4888  226.89
  4910.4  229.33  4943.3   229.7  4993.4  226.56  4997.2  222.38    5000  221.88
  5003.2  222.38  5015.7  227.02  5067.5  229.61    5188  236.07  5215.9  235.07
  5250.4  237.07  5268.5  237.79  5359.9  240.36  5389.9   239.2  5649.9  241.99
  5799.9  240.69  6187.8  242.58  6286.6  242.33  6385.3  242.46  6860.5  250.99
#Mann= 10 ,-1 , 0
  3749.3      .1       0  4409.8     .16       0  4428.5      .1       0
  4997.2     .07       0  5003.2      .1       0  5250.4     .05       0
  5268.5      .1       0  6187.8     .08       0  6286.6     .05       0
  6385.3      .1       0
Bank Sta=4943.3,5067.5
XS Rating Curve= 0 ,0
Exp/Cntr=0.3,0.1

Type RM Length L Ch R = 1 ,63357   ,790,790,790
BEGIN DESCRIPTION:
Mapping XS 0f0aa469
END DESCRIPTION:
XS GIS Cut Line= 3
      2292127.47     13333213.72      2291007.71     13334297.02
      2291059.78     13336332.64
#Sta/Elev= 30
  3969.2  258.54  3989.7  257.95  4049.1  254.21  4084.3  253.65  4423.9   236.9
  4756.3  228.64  4869.4  227.97  4940.2  225.63  4975.4  226.36  4989.6  225.38
  4993.8  221.78  4996.5  221.28  4999.8  221.78  5017.9  222.92  5039.2  226.27
  5088.6  226.31  5272.5  234.01  5498.9  240.43  5876.2  241.38    5975  241.48
  6167.3  241.26  6227.3  242.39  6477.4  240.56  6864.4  241.96  6963.2  242.35
    7062  243.06  7357.6  247.53  7427.7  250.24  7477.7  248.97  7563.5  251.71
#Mann= 9 ,-1 , 0
  3969.2     .05       0  3989.7      .1       0  4993.8     .07       0
  4999.8      .1       0  5876.2     .05       0    5975      .1       0
  6864.4     .08       0  6963.2     .05       0    7062      .1       0
Bank Sta=4975.4,5039.2
XS Rating Curve= 0 ,0
Exp/Cntr=0.3,0.1

Type RM Length L Ch R = 1 ,62567   ,514,514,514
BEGIN DESCRIPTION:
UNT003 IN NURI 87.0
END DESCRIPTION:
XS GIS Cut Line= 3
      2291037.73     13332646.81      2290937.72     13333346.85
      2291037.72     13336446.89
#Sta/Elev= 30
  4268.7  254.61  4450.6   243.8  4703.1  232.68    4837  228.05  4925.3  226.04
  4965.7   224.5  4973.3  222.14  4992.9   219.7  4995.6   219.2  4998.9   219.7
  5025.9  225.84  5065.9   224.9    5296  228.43  5456.1  228.36  5646.2  232.86
  5806.3  238.61  5976.4  241.68  6216.5  241.44  6236.5  243.01  6274.4   242.1
  6373.3  241.33  6646.7  241.99  6936.9  240.35    7137  242.05  7361.9  242.29
  7460.8  243.77  7707.3  247.04  7837.3  250.87  7957.4  251.45  8077.5  254.93
#Mann= 8 ,-1 , 0
  4268.7     .05       0    4837      .1       0  4992.9     .07       0
  4998.9      .1       0  6274.4     .05       0  6373.3      .1       0
  7361.9     .05       0  7460.8      .1       0
Bank Sta=4925.3,5025.9
XS Rating Curve= 0 ,0
Exp/Cntr=0.3,0.1

Type RM Length L Ch R = 1 ,62053   ,541,541,541
BEGIN DESCRIPTION:
UNT003 IN NURI 86.0
END DESCRIPTION:
XS GIS Cut Line= 3
      2290137.73     13333296.86      2290487.72     13333546.85
      2290887.72     13335946.85
#Sta/Elev= 30
  4574.2  248.14  4783.1  237.26  4869.1   231.1  4881.4  228.94  4896.2   229.2
  4904.8  227.56  4955.1  223.67  4990.8  220.57  4993.9   218.2  4996.7   217.7
  4999.9   218.2  5006.8  218.74  5024.6  224.06  5037.3  222.82  5136.1  223.87
  5207.1  226.88  5247.6  224.92  5328.7  225.24  5683.5  235.21  5706.4  234.56
  5724.1  236.56  5888.8  240.54  6066.4  240.28    6108  240.32  6362.8   239.1
    6525  240.83  6778.4  238.04  7314.9  245.03  7415.5  246.37  7437.4  246.46
#Mann= 7 ,-1 , 0
  4574.2      .1       0  4993.9     .07       0  4999.9      .1       0
  6066.4     .05       0    6108      .1       0  7314.9     .05       0
  7415.5      .1       0
Bank Sta=4955.1,5024.6
XS Rating Curve= 0 ,0
Exp/Cntr=0.3,0.1

Type RM Length L Ch R = 1 ,61512   ,376,376,376
BEGIN DESCRIPTION:
UNT003 IN NURI 85.0
END DESCRIPTION:
XS GIS Cut Line= 3
      2290037.72      13333346.9      2290087.72     13333896.85
      2290887.71     13336296.81
#Sta/Elev= 30
    4436   247.3  4763.6  232.62  4797.4  229.81  4969.5  222.06  4978.2  222.53
  4990.9  220.94  4995.8  216.32  4998.5  215.82  5001.8  216.32  5009.3  216.47
  5040.9  223.25  5072.5  222.02  5083.1  222.92  5104.2   221.5  5146.3  224.57
  5293.9  224.21  5378.2  226.96  5388.8  228.26  5757.7  237.75  5915.7  237.13
  6065.6  238.15  6315.9  237.51  6481.9  238.13  6634.8  239.51  6891.9   244.6
  7002.7  245.84  7017.4  246.31  7122.5   246.7    7288  248.65    7518  251.85
#Mann= 15 ,-1 , 0
    4436      .1       0  4763.6     .05       0  4969.5      .1       0
  4995.8     .07       0  5001.8      .1       0  5915.7     .05       0
  6065.6      .1       0  6315.9     .16       0  6481.9      .1       0
  6634.8     .05       0  6891.9      .1       0  7002.7     .05       0
  7017.4      .1       0  7122.5     .05       0    7288      .1       0
Bank Sta=4978.2,5040.9
XS Rating Curve= 0 ,0
Exp/Cntr=0.3,0.1

Type RM Length L Ch R = 1 ,61136   ,548,548,548
BEGIN DESCRIPTION:
Mapping XS dbf58059
END DESCRIPTION:
XS GIS Cut Line= 4
      2289971.25      13333338.7      2289757.71     13334005.35
      2290117.09     13334645.98      2290720.97     13336332.67
#Sta/Elev= 30
  4078.4  247.85    4486  232.12    4687     227    4791   225.4  4905.9   221.2
  4940.7  223.38  4995.4  215.43  4998.1  214.93  5001.4  215.43  5008.6  216.01
  5014.3  222.01    5052  220.76  5079.4  223.43  5182.1  223.13  5529.7  230.62
  5647.5     230  5772.3  232.21  6087.5  238.95    6226  239.84    6332  241.17
    6438   240.7  6543.9  241.95  6861.9  245.35  6967.9   246.3  7003.2  246.75
  7073.8  247.94  7179.8   249.1  7272.4  250.59  7285.8  250.98  7304.5  251.23
#Mann= 17 ,-1 , 0
  4078.4      .1       0    4687     .08       0    4791      .1       0
  4995.4     .07       0  5001.4      .1       0  5772.3     .05       0
    6226     .16       0    6332      .1       0    6438     .16       0
  6543.9      .1       0  6861.9     .08       0  6967.9     .05       0
  7003.2     .08       0  7073.8     .05       0  7179.8      .1       0
  7272.4     .08       0  7285.8      .1       0
Bank Sta=4940.7,5079.4
XS Rating Curve= 0 ,0
Exp/Cntr=0.3,0.1

Type RM Length L Ch R = 1 ,60588   ,747,747,747
BEGIN DESCRIPTION:
Mapping XS d0d2b349
END DESCRIPTION:
XS GIS Cut Line= 3
      2289950.43     13333312.62      2289387.92     13334312.65
      2290190.01      13336406.4
#Sta/Elev= 30
  3558.7  247.94  3609.4   247.7  3674.5  243.95  3960.7  235.12  4470.5  226.55
    4482  226.23  4581.9  225.87  4693.3   223.4  4881.9   220.9  4892.6     219
  4956.9  220.36    4972  219.93    4999  213.33  5001.8  212.83    5005  213.33
  5010.4  217.55  5032.1  220.88  5136.2  223.49  5330.4  222.95  5499.9  225.18
  5792.2  236.72  6190.8  239.48  6250.9  239.67  6297.7  239.77  6505.8  241.58
  6511.6  241.67  6618.5  243.33  6725.5  244.83    6864  247.74  6948.2  248.57
#Mann= 15 ,-1 , 0
  3558.7      .1       0  4470.5     .08       0    4482      .1       0
  4581.9     .08       0  4693.3      .1       0    4999     .07       0
    5005      .1       0  6190.8     .05       0  6250.9      .1       0
  6297.7     .05       0  6505.8     .16       0  6511.6     .05       0
  6618.5      .1       0  6725.5     .05       0    6864      .1       0
Bank Sta=4956.9,5032.1
XS Rating Curve= 0 ,0
Exp/Cntr=0.3,0.1

Type RM Length L Ch R = 1 ,59841   ,570,570,570
BEGIN DESCRIPTION:
UNT003 IN NURI 84.0
END DESCRIPTION:
XS GIS Cut Line= 3
      2289937.71     13333246.86      2288837.72     13334846.85
      2289187.73     13336396.89
#Sta/Elev= 30
  3063.6  249.36  3372.8  242.28  3495.2   237.9  4219.6   224.2    4337  222.13
    4492  219.99  4520.2  219.98  4696.1  222.42  4847.5  221.12  4932.4  217.95
  4955.9  219.42  4976.8  218.03  4994.8  212.44  4997.5  211.94  5000.8  212.44
  5002.2  214.08  5024.3  215.25  5029.4  218.12  5066.7   219.8  5120.9  220.84
  5148.8  223.28  5169.3  222.08  5189.8  223.85  5212.5  223.09  5476.8  232.32
  5605.2   233.6  5732.6  234.13  5856.1  233.32  5989.4  234.92  6594.3  248.82
#Mann= 9 ,-1 , 0
  3063.6      .1       0  4219.6     .08       0    4337      .1       0
    4492     .05       0  4520.2      .1       0  4994.8     .07       0
  5000.8      .1       0  5605.2     .08       0  5732.6      .1       0
Bank Sta=4955.9,5066.7
XS Rating Curve= 0 ,0
Exp/Cntr=0.3,0.1
