HEC-RAS study PENITAS CREEK.prj: PENITAS CREEK Base Level Engineering

--- PENITAS CREEK.g01 (geometry) --- (continued)

Type RM Length L Ch R = 1 ,73225   ,494,494,494
BEGIN DESCRIPTION:
PENITAS CREEK 127.0
END DESCRIPTION:
XS GIS Cut Line= 3
      2280087.73     13186946.86      2279837.72     13186646.85
      2279637.75     13186546.87
#Sta/Elev= 30
  4599.1  250.87  4602.4  250.87  4606.3   252.9  4634.9  253.49  4684.4  249.78
  4755.3   249.4  4811.9  248.06  4833.4  246.72  4840.6  245.42  4854.9  244.08
  4861.4  244.32  4869.2  242.59  4875.7  242.47  4883.5  240.42  4897.9  239.12
  4904.4  237.74  4918.7  236.26  4953.8  236.37  4968.1  235.08  4982.5   235.8
  4986.4  235.03    5009  235.01  5011.7  234.51  5020.4  236.56    5026  238.68
  5042.7  242.54  5065.1  244.93  5101.4   246.7  5115.4  246.68  5213.2  251.32
#Mann= 3 ,-1 , 0
  4599.1     .16       0  4904.4     .07       0    5026     .16       0
Bank Sta=4897.9,5026
XS Rating Curve= 0 ,0
Exp/Cntr=0.3,0.1

Type RM Length L Ch R = 1 ,72731   ,508,508,508
BEGIN DESCRIPTION:
PENITAS CREEK 126.0
END DESCRIPTION:
XS GIS Cut Line= 3
      2280487.71     13186796.84      2280187.72     13186396.85
      2279987.74     13186196.87
#Sta/Elev= 30
  4503.9  249.49  4511.2  249.72  4517.4   248.5  4553.9   247.8    4582  247.75
  4611.2  246.98  4617.4  247.39  4640.3  247.43  4717.4  246.03  4761.2  244.48
  4890.3  243.09  4896.6  241.36  4903.9  240.09  4925.8  239.14    4932  236.88
  4946.6  236.39  4967.4  234.85    4982  234.39  4990.3  234.65  4996.3  233.43
  5000.8  234.37    5018  234.59  5060.4  236.97  5088.7  239.49  5102.9  242.36
    5117  244.17  5159.4   245.7  5201.9  246.62  5244.3  248.34  5286.7  249.09
#Mann= 3 , 0 , 0
  4503.9     .16       0    4932     .07       0  5060.4     .16       0
Bank Sta=4932,5060.4
XS Rating Curve= 0 ,0
Exp/Cntr=0.3,0.1

Type RM Length L Ch R = 1 ,72223   ,452,452,452
BEGIN DESCRIPTION:
PENITAS CREEK 125.0
END DESCRIPTION:
XS GIS Cut Line= 3
      2280697.57     13186546.67      2280537.72     13186346.85
      2280237.73     13185896.87
#Sta/Elev= 30
  4772.4   245.9  4878.6  245.88  4950.7  241.92  4957.1  237.36  4964.3  235.02
  4971.5  234.66  4977.9  234.07  4985.9  230.28    5000   228.5  5006.7  229.14
  5014.7  232.08  5035.8  233.61  5064.3   232.9  5208.6   236.2  5237.1  238.46
  5244.6  239.98  5273.2  239.79  5288.2  241.86  5330.3  244.78  5388.8  246.22
  5432.4  248.35  5438.4  249.69  5489.5  250.27  5504.5  251.37  5510.5  249.31
  5519.5  249.94  5525.6  248.88  5555.6  251.36  5561.6  250.75  5569.1  252.17
#Mann= 4 ,-1 , 0
  4772.4     .16       0  4971.5     .07       0  5035.8     .16       0
  5569.1      .1       0
Bank Sta=4977.9,5035.8
XS Rating Curve= 0 ,0
Exp/Cntr=0.3,0.1

Type RM Length L Ch R = 1 ,71771   ,522,522,522
BEGIN DESCRIPTION:
PENITAS CREEK 124.0
END DESCRIPTION:
XS GIS Cut Line= 3
      2281030.06     13186368.46      2280937.72     13186146.85
      2280487.68     13185746.82
#Sta/Elev= 30
  4768.1  243.93  4786.6  244.42  4856.5  243.53  4863.5  242.56  4932.3  240.26
  4940.5  238.75    4954  238.39  4964.3  235.48  4969.7  236.79  4975.7  235.35
 4977.05  234.84  4998.7  229.37  5005.5  230.57  5029.5  231.44  5050.4   231.1
  5064.6  232.03  5072.1  233.08 5077.95  234.87  5078.8   233.9  5086.4  236.89
  5128.6  238.94  5135.7  236.44  5142.4  239.65  5149.9  240.24  5227.7   243.1
  5319.7  245.28  5411.6  246.26  5560.5   249.5  5596.5  251.43  5610.3  251.13
#Mann= 3 ,-1 , 0
  4768.1     .16       0  4975.7     .07       0 5077.95     .16       0
#XS Ineff= 2 , 0
       0                 5127.25       0     239
Permanent Ineff=
       F       T
Bank Sta=4977.05,5077.95
XS Rating Curve= 0 ,0
Exp/Cntr=0.3,0.1

Type RM Length L Ch R = 1 ,71249   ,454,454,454
BEGIN DESCRIPTION:
PENITAS CREEK 123.0
END DESCRIPTION:
XS GIS Cut Line= 5
      2281522.49     13187027.44      2281374.91     13186372.03
      2281387.93     13185898.94      2281387.93     13185790.43
      2280836.72     13184996.16
#Sta/Elev= 30
  3923.1  258.05    4012  254.44  4017.1   255.4  4281.8   246.9  4594.9  239.88
  4600.1   237.8  4620.1  237.97  4630.1  234.72  4670.1   231.4  4710.1  231.46
  4750.2  235.21  4760.2   238.8  4770.2  238.89  4830.2  237.55  4890.2  234.25
  4900.2  234.83 4904.96  233.03  4930.2  231.14  4960.2  231.28    5000  227.56
  5003.2  228.06  5010.3   232.9  5020.3  238.41  5170.3  242.86    5471  243.31
  5609.7  245.97  5660.6  246.74  5667.9   245.9  5848.4  248.83  6143.5  255.55
#Mann= 5 ,-1 , 0
  3923.1     .16       0 4904.96     .07       0  5010.3     .16       0
    5471     .16       0  5609.7      .1       0
#XS Ineff= 2 , 0
       0 4761.38  238.74               0
Permanent Ineff=
       T       F
Bank Sta=4904.96,5010.3
XS Rating Curve= 0 ,0
Exp/Cntr=0.3,0.1

Type RM Length L Ch R = 1 ,70795   ,396,396,396
BEGIN DESCRIPTION:
PENITAS CREEK 122.0
END DESCRIPTION:
XS GIS Cut Line= 3
      2281990.82     13186564.73       2281934.4     13186165.39
      2281044.71     13184841.71
#Sta/Elev= 30
    4394  254.99  4525.8  249.91  4553.4  250.11  4662.9  246.48  4694.8  244.04
  4785.7  242.03  4879.9   237.1  4887.9  235.92    4894  232.22  4902.9  231.65
  4908.9  234.93    4916  234.65 4920.45  232.06  4923.9  229.98  4938.9  228.35
  4988.3  227.65  4995.7  225.44  5016.9  226.87  5031.9  231.04    5038  230.37
 5041.32  232.06  5046.9  234.13  5067.9  235.58  5082.9  235.03  5103.9  237.07
  5232.9  241.28  5712.3  242.94  5721.6  242.98  5961.9  246.53  6392.2  262.48
#Mann= 5 ,-1 , 0
    4394     .16       0  4923.9     .07       0 5041.32     .16       0
  5712.3     .16       0  5721.6      .1       0
#XS Ineff= 2 , 0
       0 4909.33  234.95               0
Permanent Ineff=
       T       F
Bank Sta=4920.45,5041.32
XS Rating Curve= 0 ,0
Exp/Cntr=0.3,0.1

Type RM Length L Ch R = 1 ,70399   ,375,375,375
BEGIN DESCRIPTION:
PENITAS CREEK 121.0
END DESCRIPTION:
XS GIS Cut Line= 3
      2282237.72     13186246.82      2282187.72     13185896.85
      2281087.72     13184696.85
#Sta/Elev= 30
  4662.7  248.84    4693   249.7  4703.1     248  4965.7  234.73 4977.29  231.37
  4985.9  224.22  4995.8  222.94  5019.6  225.11  5023.3  227.35  5030.1   228.2
  5065.9  229.09  5072.6  230.67  5094.2  233.55  5157.7  234.97  5200.3  237.21
  5207.1  236.74    5257  239.09  5313.7  240.41    5540  241.11  5554.2  240.29
  5589.4  240.94  5660.3     240    5717  240.28  5908.2  242.76  6155.7  247.82
  6360.8  255.34  6502.6  262.12  6608.6  266.43    6637  266.66  6644.1   267.6
#Mann= 4 ,-1 , 0
  4662.7     .16       0 4977.29     .07       0  5072.6     .16       0
  6644.1     .05       0
Bank Sta=4977.29,5072.6
XS Rating Curve= 0 ,0
Exp/Cntr=0.3,0.1

Type RM Length L Ch R = 1 ,70024   ,403,403,403
BEGIN DESCRIPTION:
PENITAS CREEK 120.0
END DESCRIPTION:
XS GIS Cut Line= 3
      2282459.57     13186525.63      2282520.33     13185683.62
      2281504.68     13184633.25
#Sta/Elev= 30
  4242.9  259.29  4512.4   251.4  4682.8  242.78  4692.8   241.4  4722.9  240.62
    4773  237.13  4813.1  236.91  4840.3  233.52 4898.27  230.84  4973.6   227.6
  4993.4  225.22  5033.7  227.79    5039  230.91  5043.7   235.3    5207  233.52
  5242.2  235.27  5270.5   234.7  5305.8  236.75  5341.3  236.51  5348.2  237.62
  5489.7  239.43  5765.5  239.92  5871.7  236.96  6013.2  241.34  6283.9  252.29
  6425.5  258.61    6487  261.61    6494  261.12  6515.3  262.92  6548.2  262.71
#Mann= 5 ,-1 , 0
  4242.9     .16       0 4898.27     .07       0  5033.7     .16       0
  6283.9     .08       0  6425.5      .1       0
#XS Ineff= 2 , 0
       0                 5072.54       0  235.38
Permanent Ineff=
       F       T
Bank Sta=4898.27,5039
XS Rating Curve= 0 ,0
Exp/Cntr=0.3,0.1

Type RM Length L Ch R = 1 ,69621   ,463,463,463
BEGIN DESCRIPTION:
PENITAS CREEK 119.0
END DESCRIPTION:
XS GIS Cut Line= 4
      2283431.81     13186352.04      2283014.98     13185877.13
      2282589.78     13185631.54       2281635.5     13184651.23
#Sta/Elev= 30
  4210.3   262.4  4514.3  252.17  4606.4  247.69  4783.8  243.57  4833.2  240.91
  4891.9  241.13  4913.4  239.49  4919.9  233.79  4934.9  232.52 4944.73  229.84
  4950.7  228.85  4993.6   225.4  5058.4  226.75  5095.8  229.73    5345  233.83
  5408.8  231.68  5557.2   231.4  5649.1     234  5684.5  233.41  5691.5  234.84
  5712.8  234.11  5804.7  238.01  5953.3  240.24    6038  239.76    6137  235.01
  6165.3  237.51  6335.1  243.64  6566.4  255.37  6598.4  256.75  6701.3  261.65
#Mann= 5 ,-1 , 0
  4210.3     .16       0  4950.7     .07       0  5095.8     .16       0
  6566.4     .08       0  6598.4      .1       0
#XS Ineff= 2 , 0
       0                 5290.16       0  233.51
Permanent Ineff=
       F       T
Bank Sta=4944.73,5095.8
XS Rating Curve= 0 ,0
Exp/Cntr=0.3,0.1

Type RM Length L Ch R = 1 ,69158   ,881,881,881
BEGIN DESCRIPTION:
PENITAS CREEK 118.0
END DESCRIPTION:
XS GIS Cut Line= 4
      2283644.47     13186243.52      2283067.21     13185488.31
      2282772.07     13185388.48      2281917.04     13184598.55
#Sta/Elev= 30
  3812.3  259.98  4093.2  251.12    4114  249.35  4163.9  248.99    4407  241.04
  4785.9  235.11    4812   230.2  4817.3  234.21  4825.7   234.1  4836.2  232.91
  4843.5  229.91  4848.7  231.19  4857.3  230.64 4865.76  228.46  4867.9  227.57
  4937.8  226.65  5005.7  222.07  5008.9  222.57 5013.95  228.36  5015.7  230.93
  5199.1  228.97  5382.8  230.83    5461  227.46  5595.4  232.63  5679.9  232.41
  5779.1  235.45  5800.7  234.73  5977.6  244.27  6126.2  250.21  6238.5  257.37
#Mann= 4 ,-1 , 0
  3812.3     .16       0  4867.9     .07       0  5008.9     .16       0
  6238.5      .1       0
#XS Ineff= 2 , 0
       0 4818.13  234.46 5038.86       0  230.77
Permanent Ineff=
       T       T
Bank Sta=4865.76,5013.95
XS Rating Curve= 0 ,0
Exp/Cntr=0.3,0.1

Type RM Length L Ch R = 1 ,68277   ,557,557,557
BEGIN DESCRIPTION:
PENITAS CREEK 117.0
END DESCRIPTION:
XS GIS Cut Line= 3
      2283787.71     13186146.84      2283297.24      13185110.7
      2283193.08     13184173.23
#Sta/Elev= 30
  3665.4  258.96  3747.8  255.01  4019.4  246.19  4107.9  242.32  4130.1  242.43
  4287.6  236.95  4406.9  234.03    4462  231.59  4588.9  229.82  4716.4  226.45
  4782.8  225.95    4876  226.63  4936.4  225.48  4942.3  224.74  4966.6  223.19
  4996.5  219.61  5016.9  221.73  5026.9  221.85  5032.9  223.83  5037.9  224.03
 5039.31  225.42    5047  228.64  5057.1  230.38  5077.2  231.31  5318.7  237.35
  5389.1   237.5  5550.1  240.52  5576.2   242.5  5640.7  244.18    5755  249.38
#Mann= 3 ,-1 , 0
  3665.4     .16       0  4942.3     .07       0  5037.9     .16       0
Bank Sta=4936.4,5039.31
XS Rating Curve= 0 ,0
Exp/Cntr=0.3,0.1

Type RM Length L Ch R = 1 ,67720   ,846,846,846
BEGIN DESCRIPTION:
PENITAS CREEK 116.0
END DESCRIPTION:
XS GIS Cut Line= 3
      2283887.72     13186146.81      2283787.72     13184946.85
      2283487.72     13183846.84
#Sta/Elev= 30
  3823.9  258.97  4395.8  238.21    4747  232.49  4837.4  229.23  4897.6   224.9
 4901.97  223.44  4907.6  222.52  4937.7  220.25  4977.8  220.33  4997.7  217.73
  5007.9  220.38    5018  222.86  5025.5   224.4  5050.5  224.63    5225  224.62
    5339  227.95  5387.3  227.88  5525.5  233.28  5546.3  232.76  5575.6  234.98
  5615.4  236.62  5620.6  235.86  5660.3  239.85    5681  239.86  5784.7   246.5
    5795  245.24  5826.1  247.92  5950.5  252.83  6054.2  259.83  6168.2  264.94
#Mann= 3 ,-1 , 0
  3823.9     .16       0  4907.6     .07       0  5007.9     .16       0
#XS Ineff= 2 , 0
       0                 5125.91       0  225.54
Permanent Ineff=
       F       T
Bank Sta=4901.97,5018
XS Rating Curve= 0 ,0
Exp/Cntr=0.3,0.1

Type RM Length L Ch R = 1 ,66874   ,637,637,637
BEGIN DESCRIPTION:
Mapping XS 4d77f0eb
END DESCRIPTION:
XS GIS Cut Line= 3
       2283991.7     13185952.67      2284178.32     13184863.31
      2283957.08     13183991.37
#Sta/Elev= 30
  3549.9  252.02  3981.9  236.49  4103.7  234.33    4564  231.37  4718.5  226.36
  4775.3   225.7  4841.4  221.63  4877.2  221.28  4882.4  220.78  4899.1  218.12
  4909.4  219.01    4930  217.88  4950.7  219.61  4981.6  216.75  5000.1   216.2
  5005.3  217.07  5012.3  215.63 5036.36  221.25  5041.1  223.24  5064.1  222.89
  5087.2  226.05  5229.2  233.25  5245.9  235.67  5251.1  235.16    5292  239.67
  5327.8  242.07  5445.6  247.67  5486.5  248.45  5538.7  251.18  5554.7  253.08
#Mann= 3 ,-1 , 0
  3549.9     .16       0  4882.4     .07       0 5036.36     .16       0
Bank Sta=4877.2,5036.36
XS Rating Curve= 0 ,0
Exp/Cntr=0.3,0.1

Type RM Length L Ch R = 1 ,66237   ,346,346,346
BEGIN DESCRIPTION:
PENITAS CREEK 115.0
END DESCRIPTION:
XS GIS Cut Line= 3
      2284087.73     13185796.82      2284608.01     13184503.06
      2284413.35      13184070.5
#Sta/Elev= 30
  3799.4  245.86  3945.8  239.97  4068.8  236.68  4082.9   237.4  4090.4   236.4
  4122.7   235.7  4537.1  230.81  4674.1  230.57  4683.2  231.26  4692.9  230.43
  4769.4  230.27  4805.8  228.98  4883.7  223.09  4913.3  222.16  4920.3  220.33
  4931.1  221.33  4937.5  220.09  4942.9  217.52  4961.7  216.14    4967  216.44
  4974.2  219.54  4996.4  213.26  5020.8  215.43  5038.9   218.6  5092.8  219.45
  5275.9  227.43  5500.7  234.73  5540.6  234.89  5552.5  236.24  5668.2  240.22
#Mann= 4 ,-1 , 0
  3799.4     .16       0  4974.2     .07       0  5038.9     .16       0
  5668.2     .05       0
#XS Ineff= 1 ,-1
 4886.01 4974.09  219.64
Permanent Ineff=
       T
Bank Sta=4974.2,5038.9
XS Rating Curve= 0 ,0
Exp/Cntr=0.3,0.1

Type RM Length L Ch R = 1 ,65891   ,423,423,423
BEGIN DESCRIPTION:
PENITAS CREEK 114.0
END DESCRIPTION:
XS GIS Cut Line= 3
      2284386.66     13185800.79      2284824.61     13184933.97
      2284955.22     13184203.63
#Sta/Elev= 30
    3799  241.29  3877.6  238.06  4016.9  237.99  4496.2  227.07    4563  226.53
  4621.3  228.76  4702.4  229.62  4763.7   228.4  4777.4   226.7  4797.7  229.11
  4819.7  226.49  4838.3  227.14  4919.6  224.07  4960.3  220.98 4963.81  218.88
  4986.2  213.01  4991.2  213.62  5000.6     212    5011  212.59  5021.2  216.97
  5031.4  217.46  5061.8  216.74    5133  218.69  5143.1  216.21  5157.7  214.78
  5173.6  216.13  5183.7  219.06  5275.5  224.45  5441.9  229.92  5512.1  230.68
#Mann= 4 ,-1 , 0
    3799     .16       0 4963.81     .07       0  5031.4     .16       0
  5512.1      .1       0
#XS Ineff= 2 , 0
       0                 5133.68       0  218.71
Permanent Ineff=
       F       T
Bank Sta=4963.81,5031.4
XS Rating Curve= 0 ,0
Exp/Cntr=0.3,0.1

Type RM Length L Ch R = 1 ,65468   ,845,845,845
BEGIN DESCRIPTION:
PENITAS CREEK 113.0
END DESCRIPTION:
XS GIS Cut Line= 3
      2285037.71      13185746.9      2285237.72     13184546.85
      2285187.72     13184146.86
#Sta/Elev= 30
  3795.8  245.36  3884.6  242.74  3927.6  239.93  3958.1  239.77  4079.7  235.13
  4170.9  232.76  4249.5   229.5  4262.2  227.93  4302.7  227.15  4444.7  220.68
  4475.1  220.73  4485.2  219.52  4748.8  217.82    4797  218.87  4819.8  218.39
  4840.1  216.71  4857.8  217.38  4961.7  215.13  4984.5  213.12  4992.1  210.06
    5002  209.13  5042.6  214.44  5050.2  217.99  5055.2  218.89  5082.9  221.49
  5113.2  220.07  5123.3  224.12  5183.7   227.3  5244.2  229.34  5415.5  232.44
#Mann= 3 ,-1 , 0
  3795.8     .16       0  4819.8     .07       0  5050.2     .16       0
Bank Sta=4819.8,5055.2
XS Rating Curve= 0 ,0
Exp/Cntr=0.3,0.1

Type RM Length L Ch R = 1 ,64623   ,527,527,527
BEGIN DESCRIPTION:
PENITAS CREEK 112.0
END DESCRIPTION:
XS GIS Cut Line= 4
      2285402.27     13185813.84      2285693.08     13185319.04
      2285810.26     13184746.12      2285728.05     13184110.02
#Sta/Elev= 30
  4248.3  243.25  4271.4  241.68    4330  240.83  4644.4  230.77  4687.4   229.8
    4703  230.56  4724.5  228.53  4813.2  226.51  4820.2  224.83  4870.4  222.21
  4885.7  219.72  4906.1  219.99  4915.7  218.09  4920.8  217.41  4926.5  214.98
  4997.7  209.72  5016.7  210.64  5038.8  213.82    5049  214.15  5110.3  214.44
  5117.6   213.5  5161.3  213.36  5212.3  215.16  5314.4  215.23  5396.1  217.99
  5486.9  223.07  5567.6  226.13  5648.3  227.31  5870.1   227.9  6048.4  231.19
#Mann= 5 ,-1 , 0
  4248.3     .16       0  4920.8     .07       0  5396.1     .16       0
  6048.4      .1       0  6048.4      .1       0
Bank Sta=4915.7,5396.1
XS Rating Curve= 0 ,0
Exp/Cntr=0.3,0.1

Type RM Length L Ch R = 1 ,64096   ,63,63,63
BEGIN DESCRIPTION:
Mapping XS 2e64df63
END DESCRIPTION:
XS GIS Cut Line= 2
      2286131.44     13185536.02      2286122.77     13184581.56
#Sta/Elev= 30
  4432.4  232.56  4571.6  228.53  4621.6  226.44  4661.6  224.31  4681.6  222.05
  4711.6  220.98  4721.6  221.53  4731.6  220.03  4751.6  218.37  4791.6  217.26
  4801.6   215.3  4811.6  214.88  4831.6  215.75  4841.6  218.66  4851.6   219.8
  4861.6  218.51  4871.6  216.83  4881.6   213.7  4901.6  208.78  5021.6  208.86
  5038.6  208.64  5041.3  208.14  5044.6  208.64  5081.6  209.12  5091.6  211.85
  5101.6  213.55  5111.6  217.11  5121.6  217.93  5241.6  224.41  5386.9  225.17
#Mann= 4 ,-1 , 0
  4432.4     .16       0  4871.6     .07       0  5121.6     .16       0
  5386.9     .05       0
#XS Ineff= 1 ,-1
  4717.1 4849.74  219.69
Permanent Ineff=
       T
Bank Sta=4861.6,5121.6
XS Rating Curve= 0 ,0
Exp/Cntr=0.3,0.1

Type RM Length L Ch R = 1 ,64033   ,96,96,96
BEGIN DESCRIPTION:
PENITAS CREEK 111.0
END DESCRIPTION:
XS GIS Cut Line= 2
      2286183.31     13185488.78      2286193.73     13184587.74
#Sta/Elev= 30
  4486.4  230.71  4558.3  228.79  4578.3  227.68  4588.3  226.22  4608.3  226.67
  4638.3  225.47  4658.3  223.34  4678.3  222.19  4768.3  218.85  4788.3  217.16
  4798.3  215.27  4818.1  214.12  4838.3  216.88  4848.3  220.17  4858.4  220.71
  4868.4  220.35  4878.4  219.11  4898.4  218.33  4928.4  218.31  4958.4  219.21
  5118.4  222.07  5168.4  222.13  5228.4     224  5238.4  224.47  5248.4  228.88
  5258.4  229.81  5268.4  228.82  5278.4  229.43  5296.9   224.8  5387.5  224.91
#Mann= 4 ,-1 , 0
  4486.4     .16       0  4878.4     .07       0  4958.4     .16       0
  5387.5     .05       0
#XS Ineff= 2 , 0
       0 4858.03  220.69               0
Permanent Ineff=
       T       F
Bank Sta=4878.4,4958.4
XS Rating Curve= 0 ,0
Exp/Cntr=0.3,0.1

Type RM Length L Ch R = 1 ,63937   ,272,272,272
BEGIN DESCRIPTION:
Mapping XS d662aeef
END DESCRIPTION:
XS GIS Cut Line= 2
      2286270.33      13185553.4      2286257.32     13184581.48
#Sta/Elev= 30
  4458.4  231.75    4625  226.87    4635  225.08    4655  223.08    4705  220.35
    4725  221.21    4735  222.76    4765  225.17    4775  222.34    4785  220.77
    4795  217.65    4865  213.35    4875  213.91    4895  212.36    4945  211.22
    4975  209.43    4985  208.04    5015  207.18  5023.5  208.16  5025.5  206.99
  5028.2  206.49    5085  211.07    5115  217.03    5165  218.79    5185  220.95
    5205  220.06    5215  222.66    5235  223.67    5285  224.61  5430.4  224.62
#Mann= 4 ,-1 , 0
  4458.4     .16       0    4945     .07       0    5085     .16       0
  5430.4     .05       0
Bank Sta=4945,5085
XS Rating Curve= 0 ,0
Exp/Cntr=0.3,0.1

Type RM Length L Ch R = 1 ,63665   ,354,354,354
BEGIN DESCRIPTION:
PENITAS CREEK 110.0
END DESCRIPTION:
XS GIS Cut Line= 3
      2286533.46     13185606.29      2286545.96     13185350.05
      2286458.46     13184656.29
#Sta/Elev= 30
  4482.8  229.79  4502.3  228.36  4512.3  228.43  4522.3   227.2  4592.4  225.38
  4602.4   223.6  4692.5  219.43  4722.5  217.23  4766.5  216.72  4772.8  215.67
  4782.9  215.75    4793  214.01  4833.3  212.82  4853.4  213.37  4893.8   210.6
    4922  209.41    4927  210.09  4984.5  207.55  4994.3   206.1  5014.7  207.26
  5024.8  208.78    5055  209.12  5065.1  210.53  5075.2   211.4  5082.5  213.21
  5087.6  212.75  5155.8   218.3  5216.3  221.31  5337.2  223.45  5438.6  222.88
#Mann= 4 ,-1 , 0
  4482.8     .16       0  4893.8     .07       0  5065.1     .16       0
  5438.6      .1       0
Bank Sta=4927,5065.1
XS Rating Curve= 0 ,0
Exp/Cntr=0.3,0.1

Type RM Length L Ch R = 1 ,63311   ,656,656,656
BEGIN DESCRIPTION:
PENITAS CREEK 109.0
END DESCRIPTION:
XS GIS Cut Line= 4
      2286883.46     13185668.83      2286877.21     13185400.05
      2286808.46     13184837.55      2286577.22     13184593.82
#Sta/Elev= 30
  4491.9  227.77  4673.9  221.23  4793.4  215.65  4798.5  216.04  4844.6  213.15
  4864.7  209.98  4874.8  210.12    4880  209.19    4885  210.29 4901.93  209.09
    4905  207.91  4935.2  206.64  4961.5  206.89  4985.6  205.46  4995.4  203.44
  5015.8  206.44  5048.1  207.17  5076.3  209.06  5187.1  213.28  5297.9  220.51
  5342.4  220.77  5349.7  220.06  5413.2  219.84  5434.6  218.67    5484  218.26
  5519.6  218.74  5533.7  219.75  5540.6  219.01  5597.2  219.31  5663.4  220.61
#Mann= 4 ,-1 , 0
  4491.9     .16       0    4905     .07       0  5076.3     .16       0
  5663.4      .1       0
Bank Sta=4901.93,5076.3
XS Rating Curve= 0 ,0
Exp/Cntr=0.3,0.1

Type RM Length L Ch R = 1 ,62655   ,423,423,423
BEGIN DESCRIPTION:
PENITAS CREEK 108.0
END DESCRIPTION:
XS GIS Cut Line= 3
      2287408.46     13185675.04      2287464.71     13185425.05
      2287464.71     13184700.99
#Sta/Elev= 30
  4405.8  228.47  4513.9  224.11  4519.1  224.79  4557.2  223.38  4578.2  221.59
    4654  218.89  4658.5  217.98  4780.2  213.07  4810.2  211.12  4860.2  209.54
  4870.2  208.58  4910.2  207.05  4950.2  206.49  4980.2  203.62  4990.2  203.45
  4997.2  200.28    5000  199.78  5003.2  200.28  5010.2  203.58  5020.2  204.72
  5040.2  203.74  5060.2  203.88  5070.2  204.19  5080.2  205.91  5090.2  206.71
  5100.2  208.11  5120.2  209.46  5250.2  216.21  5320.2  218.67  5386.1  219.33
#Mann= 3 , 0 , 0
  4405.8     .16       0  4950.2     .07       0  5090.2     .16       0
Bank Sta=4950.2,5090.2
XS Rating Curve= 0 ,0
Exp/Cntr=0.3,0.1

Type RM Length L Ch R = 1 ,62232   ,417,417,417
BEGIN DESCRIPTION:
PENITAS CREEK 107.0
END DESCRIPTION:
XS GIS Cut Line= 3
       2287789.7     13185612.58      2287845.96     13185387.55
      2287920.93     13184831.54
#Sta/Elev= 30
  4544.3  221.07  4679.7  217.48  4726.1  217.09  4762.2  214.98  4779.1  214.62
  4824.6  211.55  4857.7  210.22  4867.8  209.08  4908.1   206.6  4948.5  205.12
  4980.2  205.49  4988.9  203.51  4995.9  198.55  4998.7  198.05  5001.9  198.55
    5009  201.56  5019.1  202.96  5029.2  203.33  5039.3  205.05  5047.9  205.34
  5052.9  204.76  5069.6  204.49  5109.9   205.3  5140.2  207.78  5170.5  209.38
  5190.7  211.23  5198.4  211.61  5203.4  211.25  5271.1  215.19  5337.3  216.18
#Mann= 4 ,-1 , 0
  4544.3     .16       0  4980.2     .07       0  5039.3     .16       0
  5337.3     .16       0
Bank Sta=4980.2,5039.3
XS Rating Curve= 0 ,0
Exp/Cntr=0.3,0.1

Type RM Length L Ch R = 1 ,61815   ,372,372,372
BEGIN DESCRIPTION:
PENITAS CREEK 106.0
END DESCRIPTION:
XS GIS Cut Line= 3
      2288145.95     13185656.32      2288283.46     13185387.55
       2288302.2      13184881.6
#Sta/Elev= 30
  4471.2  217.53  4493.1  216.97  4636.6  216.24  4725.5  215.09  4753.3  214.21
  4793.8  212.24  4803.8  211.12  4833.8  209.82  4873.9  207.26  4903.9  204.73
  4923.9  203.68  4933.9  203.68  4953.9   202.2  4963.9  203.29  4973.9  202.52
  4983.9  202.03    4994  198.89  5003.7  198.05    5007  198.55    5014  203.24
  5026.2  203.35    5034   202.2    5054  202.32    5074  203.94    5094  204.56
    5134   207.4  5144.1  207.45  5154.1   208.9  5204.1  212.38  5279.4  214.93
#Mann= 4 ,-1 , 0
  4471.2     .16       0  4973.9     .07       0    5014     .16       0
  5279.4      .1       0
Bank Sta=4963.9,5014
XS Rating Curve= 0 ,0
Exp/Cntr=0.3,0.1

Type RM Length L Ch R = 1 ,61443   ,316,316,316
BEGIN DESCRIPTION:
PENITAS CREEK 105.0
END DESCRIPTION:
XS GIS Cut Line= 2
      2288658.46     13185718.84      2288658.46     13185006.34
#Sta/Elev= 30
  4478.4  213.83  4490.4   213.8  4510.4  214.55  4520.4  213.77  4530.4  213.66
  4600.4  214.35  4620.4  213.66  4680.4  213.56  4730.4  212.73  4790.4  210.36
  4800.4  209.33  4850.4   206.8  4860.4  205.74  4870.4  205.46  4900.4  203.31
  4940.4  201.83  4950.4  202.33  4960.4   200.7  4980.4  201.38  4990.4   200.7
  5000.1     198  5003.4   198.5  5010.4  201.57  5020.4  203.17  5060.4  202.68
  5080.4  203.35  5120.4  206.21  5130.4  207.94  5140.4  208.72  5190.9  209.76
#Mann= 4 ,-1 , 0
  4478.4     .16       0  4950.4     .07       0  5020.4     .16       0
  5190.9      .1       0
Bank Sta=4950.4,5020.4
XS Rating Curve= 0 ,0
Exp/Cntr=0.3,0.1

Type RM Length L Ch R = 1 ,61127   ,629,629,629
BEGIN DESCRIPTION:
PENITAS CREEK 104.0
END DESCRIPTION:
XS GIS Cut Line= 3
      2288977.21     13185675.09      2288964.71     13184887.55
      2288852.19     13184568.77
#Sta/Elev= 30
    4545  212.31  4653.3  211.52  4773.3  211.86  4833.3   211.1  4893.3     209
  4903.3  207.41  4963.3  202.23  4973.3  201.81  4983.3  200.43  4993.3  197.62
    5003  197.03  5023.3  200.75  5033.3   200.3  5053.3  202.06  5073.3     201
  5103.3  201.39  5173.3  204.61  5223.3   202.4  5253.3   202.8  5303.3  205.86
  5364.3  206.93  5400.5  208.95  5431.4  211.44    5450  213.91  5457.1   216.3
  5471.2  214.29  5481.8  213.66  5518.9  214.72  5534.9  216.15  5670.7  219.77
#Mann= 4 ,-1 , 0
    4545     .16       0  4973.3     .07       0  5053.3     .16       0
  5670.7     .05       0
#XS Ineff= 2 , 0
       0                 5171.81       0  204.74
Permanent Ineff=
       F       T
Bank Sta=4963.3,5053.3
XS Rating Curve= 0 ,0
Exp/Cntr=0.3,0.1

Type RM Length L Ch R = 1 ,60498   ,424,424,424
BEGIN DESCRIPTION:
PENITAS CREEK 103.0
END DESCRIPTION:
XS GIS Cut Line= 4
      2289245.93     13185600.07      2289383.46     13185512.55
      2289683.46     13185000.05      2289708.46     13184656.33
#Sta/Elev= 30
  4440.6  210.46  4515.8  209.57  4546.3  208.34  4588.6  208.69  4624.8  207.89
  4677.6  207.87  4749.3  205.44  4859.4  200.03  4902.5  199.81  4939.6  200.63
  4976.7  197.58  4992.4  197.02    4998   195.6  5013.9   198.3  5035.4  200.48
  5072.6  202.93  5166.4  206.04  5250.8  209.91  5320.6  214.05  5325.6  213.68
  5371.1  215.33  5401.2     217  5421.3  218.67  5431.3  222.08  5441.3  223.92
  5451.3  220.82  5464.7  220.19  5501.5  221.41  5511.5  222.83  5542.1  223.83
#Mann= 4 ,-1 , 0
  4440.6     .16       0  4939.6     .07       0  5035.4     .16       0
  5542.1     .05       0
Bank Sta=4939.6,5035.4
XS Rating Curve= 0 ,0
Exp/Cntr=0.3,0.1

Type RM Length L Ch R = 1 ,60074   ,462,462,462
BEGIN DESCRIPTION:
PENITAS CREEK 102.0
END DESCRIPTION:
XS GIS Cut Line= 3
      2289945.96     13185581.34      2289983.46      13185056.3
       2289939.7     13184656.27
#Sta/Elev= 30
  4748.8  205.46  4793.4     205  4853.6  203.23  4903.7  200.34  4953.8  197.35
  4981.5  197.22  4993.7  195.99  4996.9  196.49    5034  198.24  5064.1  198.56
  5084.1  199.64  5104.2  199.26  5121.8   200.2  5144.3  200.46  5194.4  202.53
  5204.4  203.41  5214.5  203.28  5244.5  204.86  5365.2  208.31  5372.1  208.81
  5385.3  208.77  5445.6  210.75  5495.9  213.09  5559.6  214.72  5576.4  216.17
  5596.5  223.29  5606.6  222.34  5626.7  219.08  5636.8   218.8  5677.6  221.26
#Mann= 4 ,-1 , 0
  4748.8     .16       0  4903.7     .07       0  5084.1     .16       0
  5677.6     .05       0
Bank Sta=4903.7,5084.1
XS Rating Curve= 0 ,0
Exp/Cntr=0.3,0.1

Type RM Length L Ch R = 1 ,59612   ,738,738,738
BEGIN DESCRIPTION:
PENITAS CREEK 101.0
END DESCRIPTION:
XS GIS Cut Line= 4
      2290270.94     13185662.57      2290408.46     13185475.05
      2290414.71     13184950.05      2290152.49     13184556.72
#Sta/Elev= 30
  4622.7  204.02  4781.3  200.87  4831.5  200.68  4883.4  201.53  4943.4  198.07
    4950  197.55  4983.4  196.72  4993.2  194.19  5003.4  194.73  5013.4  196.48
  5053.5  197.65  5093.5  197.56  5113.5  196.42  5153.5  197.61  5215.9  196.87
  5323.5  198.77    5387  201.14  5444.2  204.52  5504.2  206.64  5525.2  208.22
  5612.3  211.36  5654.4  213.42  5669.4  214.91  5726.5  215.93  5732.7  215.41
  5747.5  216.78  5813.7  219.26  5828.7  220.47  5849.7  224.18    5853  223.44
#Mann= 4 ,-1 , 0
  4622.7     .16       0  4943.4     .07       0  5053.5     .16       0
    5853     .05       0
Bank Sta=4950,5053.5
XS Rating Curve= 0 ,0
Exp/Cntr=0.3,0.1

Type RM Length L Ch R = 1 ,58874   ,289,289,289
BEGIN DESCRIPTION:
Mapping XS dd524fad
END DESCRIPTION:
XS GIS Cut Line= 3
       2290425.5     13185678.19      2290833.49     13185504.58
      2291214.53     13184790.13
#Sta/Elev= 30
  4184.4  203.44  4278.2  199.37  4325.5   196.4    4415  193.75    4460  193.71
  4512.8   194.7  4607.2   194.1  4710.7  194.91  4754.6  195.93  4783.9  194.97
  4829.2  195.56  4902.6  194.58  4918.9  195.28  4962.9  195.39  4976.5  195.25
  4984.8  194.11  4990.5  194.22    4999  192.35  5002.2  192.85  5006.8  194.97
  5012.4  194.35  5050.7  195.58  5056.2  196.02  5132.9  200.71  5220.7  204.89
  5264.6  205.34  5330.5  209.95  5339.2  211.46  5361.9  211.33  5437.5  214.17
#Mann= 3 ,-1 , 0
  4184.4     .16       0  4962.9     .07       0  5056.2     .16       0
#XS Ineff= 2 , 0
       0 4752.75  196.03               0
Permanent Ineff=
       T       F
Bank Sta=4976.5,5050.7
XS Rating Curve= 0 ,0
Exp/Cntr=0.3,0.1

Type RM Length L Ch R = 1 ,58585   ,555,555,555
BEGIN DESCRIPTION:
PENITAS CREEK 100.0
END DESCRIPTION:
XS GIS Cut Line= 4
      2290668.55     13186320.57      2290872.55     13186012.39
      2291085.23     13185621.77      2291462.79     13184866.65
#Sta/Elev= 30
    3919  206.67  4079.4  204.86    4386  192.98    4480  192.91  4495.9  189.19
  4501.8  190.89    4534  190.53  4568.2   191.3  4613.7  194.49  4636.5   197.2
  4716.2  200.41  4747.3  200.44  4819.9  194.56  4850.7  193.39  4970.9  194.32
  4976.5  194.24  4998.8  191.65  5007.2  193.67  5015.6  193.87  5021.2  194.12
  5082.7  193.71  5186.1  195.22    5351  202.47  5387.3  205.14  5468.4  207.65
  5499.1  209.54  5535.5  210.06  5552.3   212.7  5557.8  210.88  5577.6  212.95
#Mann= 4 ,-1 , 0
    3919     .16       0  4970.9     .07       0  5015.6     .16       0
  5577.6      .1       0
#XS Ineff= 2 , 0
       0 4747.56  200.54               0
Permanent Ineff=
       T       F
Bank Sta=4976.5,5021.2
XS Rating Curve= 0 ,0
Exp/Cntr=0.3,0.1

Type RM Length L Ch R = 1 ,58030   ,1167,1167,1167
BEGIN DESCRIPTION:
PENITAS CREEK 99.0
END DESCRIPTION:
XS GIS Cut Line= 5
      2290833.47     13186433.42      2291154.67     13186025.42
      2291475.85     13185717.26      2291836.09     13185352.67
      2291970.38     13185101.42
#Sta/Elev= 30
  3701.9     206  3745.6  205.61  3909.2  192.86  3965.3  189.93  4079.3  188.41
  4223.7  189.54  4236.3  187.45  4243.5  188.97  4271.8  189.86  4321.4  189.27
  4469.9   191.2  4512.3  191.04  4568.9  188.72  4611.4   192.4    4675  193.31
  4957.8  192.27  4964.8  191.67  5000.2  190.29  5014.4  191.88  5042.7  191.99
  5049.7  193.53  5056.8  192.41    5078   195.1  5085.1  194.26  5106.3  196.96
  5113.4     195  5134.6  195.69  5141.7  197.35    5170  199.41  5463.7  208.34
#Mann= 3 ,-1 , 0
  3701.9     .16       0  4964.8     .07       0  5042.7     .16       0
#XS Ineff= 2 , 0
       0 4905.18  193.01               0
Permanent Ineff=
       T       F
Bank Sta=4957.8,5042.7
XS Rating Curve= 0 ,0
Exp/Cntr=0.3,0.1

Type RM Length L Ch R = 1 ,56863   ,393,393,393
BEGIN DESCRIPTION:
Mapping XS ae27ebe0
END DESCRIPTION:
XS GIS Cut Line= 5
      2290907.25     13186485.49      2291219.77     13186359.62
      2291532.27     13186038.44      2291784.01     13185990.69
      2292013.38     13185458.37
#Sta/Elev= 30
  4362.8  204.43  4394.8  204.12  4400.2  204.74  4590.9  199.67  4701.8  199.04
  4756.9  197.81  4763.8  196.96  4813.4  195.41  4820.4  194.06  4855.9  192.51
  4884.2  190.11 4895.13  189.19  4961.9  187.38    4983  187.55  4996.9  184.54
  5004.3  186.71  5018.5  188.02  5032.6   188.3  5046.8  187.34 5071.92  189.08
    5075  189.53  5214.5  192.53    5348  191.81  5425.3   193.1  5501.3  193.21
  5734.9  198.34  5781.9  197.01  5857.9  196.46  5963.6  198.27  5983.7  197.88
#Mann= 4 ,-1 , 0
  4362.8     .16       0  4884.2     .07       0    5075     .16       0
  5983.7      .1       0
Bank Sta=4895.13,5071.92
XS Rating Curve= 0 ,0
Exp/Cntr=0.3,0.1

Type RM Length L Ch R = 1 ,56470   ,591,591,591
BEGIN DESCRIPTION:
PENITAS CREEK 98.0
END DESCRIPTION:
XS GIS Cut Line= 5
      2291427.19     13186831.32      2291664.71      13186618.8
      2291795.96     13186125.05      2292033.46      13185606.3
      2292058.47     13185475.01
#Sta/Elev= 30
  4282.6  205.02  4434.7  202.44  4569.3  198.88  4613.7     199  4644.7   197.1
  4665.4  197.32    4671  194.52  4711.2  192.64  4717.2  191.48  4746.1  190.25
  4779.2  187.24  4851.7  184.14  4893.1  186.04  4913.7   185.2  4934.4  186.67
  4946.9  186.01  4975.8   186.5  5006.6  183.63  5009.9  184.13  5022.1  187.16
  5037.9  191.31  5048.3  192.53  5089.7  193.28  5187.2  192.92  5317.2  195.82
  5443.2  195.24  5609.8  195.88  5735.2  196.71  5773.8     198  5816.4  198.08
#Mann= 3 ,-1 , 0
  4282.6     .16       0  4779.2     .07       0  5009.9     .16       0
Bank Sta=4779.2,5022.1
XS Rating Curve= 0 ,0
Exp/Cntr=0.3,0.1

Type RM Length L Ch R = 1 ,55879   ,429,429,429
BEGIN DESCRIPTION:
PENITAS CREEK 97.0
END DESCRIPTION:
XS GIS Cut Line= 3
      2291939.71      13187006.3      2292195.96     13186700.05
      2292383.41     13185631.58
#Sta/Elev= 30
  4293.8  201.77  4356.3  201.28  4405.7  198.12  4412.3  198.68    4420  196.15
  4448.7  193.16  4462.6  193.78  4469.5  192.47  4498.1  196.17    4519  193.08
  4526.7  193.51  4554.1  190.75  4604.8  190.13  4611.3  190.33  4625.6   195.1
  4726.8  197.37  4858.8   188.8  4889.3  185.88  4905.2  183.93  4950.2   184.2
  4990.8   182.7  5000.7  181.09  5011.1  182.96  5051.7  185.48  5078.3  187.19
  5173.5  187.07  5315.8  193.67  5498.4  197.16  5731.9  197.47  5777.9  198.45
#Mann= 4 ,-1 , 0
  4293.8     .16       0  4889.3     .07       0  5051.7     .16       0
  5777.9      .1       0
#XS Ineff= 2 , 0
       0                 5092.02       0  187.37
Permanent Ineff=
       F       T
Bank Sta=4889.3,5051.7
XS Rating Curve= 0 ,0
Exp/Cntr=0.3,0.1

Type RM Length L Ch R = 1 ,55450   ,520,520,520
BEGIN DESCRIPTION:
PENITAS CREEK 96.0
END DESCRIPTION:
XS GIS Cut Line= 4
      2292595.96      13186931.3      2292633.46     13186712.55
      2292733.46     13186050.05      2292789.71     13185656.29
#Sta/Elev= 30
  4519.7  197.68  4544.5  197.94  4625.7   195.8  4727.1   194.4  4828.3  189.45
  4909.2  184.47  4919.3  184.06  4936.1  182.33  4990.1  180.89  4999.9  178.24
  5004.7  177.67    5008  178.17  5010.3  181.32  5020.5  182.86  5081.1  184.24
  5111.5   184.8  5182.3     184  5232.8  185.13  5354.2  193.13  5384.5  192.62
  5403.2  192.86  5408.3  193.74  5410.7  192.69  5435.1  191.25  5549.5  191.17
  5697.7  192.56  5761.7  194.01  5778.5  193.41  5798.7  194.56  5809.4  194.42
#Mann= 4 ,-1 , 0
  4519.7     .16       0  4909.2     .07       0  5081.1     .16       0
  5809.4      .1       0
#XS Ineff= 2 , 0
       0                  5111.3       0  184.87
Permanent Ineff=
       F       T
Bank Sta=4919.3,5081.1
XS Rating Curve= 0 ,0
Exp/Cntr=0.3,0.1

Type RM Length L Ch R = 1 ,54930   ,242,242,242
BEGIN DESCRIPTION:
PENITAS CREEK 95.0
END DESCRIPTION:
XS GIS Cut Line= 3
      2293045.98     13186981.26      2293120.96      13186806.3
      2293301.93     13185820.32
#Sta/Elev= 30
    4475  198.92  4534.2  199.04  4593.8   197.7  4653.9  195.12  4667.6  195.18
  4672.5  194.12  4725.6  191.65  4730.7  194.04    4736  190.62  4807.1  187.15
    4842  184.36    4858  183.61  4878.3  184.21  4895.1  183.56  4908.8  182.18
  4929.1  182.53  4939.3  182.24  4990.1  178.16    5000  174.74  5011.5  176.55
  5020.6  179.44  5051.1   182.1  5059.5  182.74  5071.5  182.41  5081.6  184.68
  5183.3  190.27  5213.8  191.76  5264.6  192.94    5529  193.29  5667.8  194.37
#Mann= 3 ,-1 , 0
    4475     .16       0  4929.1     .07       0  5059.5     .16       0
Bank Sta=4939.3,5051.1
XS Rating Curve= 0 ,0
Exp/Cntr=0.3,0.1

Type RM Length L Ch R = 1 ,54688   ,244,244,244
BEGIN DESCRIPTION:
PENITAS CREEK 94.0
END DESCRIPTION:
XS GIS Cut Line= 3
       2293239.7     13186912.57      2293333.46     13186762.55
       2293633.1     13185907.33
#Sta/Elev= 30
  4567.3  196.75  4591.8  195.25  4670.8  191.93  4701.5  189.72  4715.6  189.55
  4813.8  183.09  4862.2   181.1  4898.6  180.27    4919   180.3  4930.4  181.07
  4962.2  180.65    4981  177.63  4986.3  177.62    4991  173.21  4993.7  172.71
  5004.6  173.62    5012  178.39  5025.7  179.53  5036.3  181.03  5048.3  181.91
  5057.5  183.43  5089.3  184.81  5130.8  187.85  5161.8  188.07  5174.1  190.02
  5254.8  192.01  5460.2  191.36  5544.9  192.11  5590.7  193.11  5650.4  193.13
#Mann= 4 ,-1 , 0
  4567.3     .16       0  4962.2     .07       0  5036.3     .16       0
  5650.4      .1       0
Bank Sta=4962.2,5036.3
XS Rating Curve= 0 ,0
Exp/Cntr=0.3,0.1

Type RM Length L Ch R = 1 ,54444   ,146,146,146
BEGIN DESCRIPTION:
Mapping XS ad812bd2
END DESCRIPTION:
XS GIS Cut Line= 3
      2293370.99     13186962.52      2293758.46     13186475.05
        2293883.     13186082.75
#Sta/Elev= 30
  4580.7  195.42  4588.9  194.98  4596.9  192.77  4603.3  193.23  4611.4  191.45
  4625.8  192.13  4632.2  190.79    4639  191.77    4653  191.57  4689.9  188.83
  4696.3  189.14  4702.9  187.88  4717.1  187.03  4795.6  184.47  4874.1  180.76
  4973.4  178.79    5002  175.47  5016.6     178  5045.5  180.63  5066.3  180.92
  5073.4  181.48  5080.7  183.53  5101.5  183.46  5130.4  184.86  5137.2  186.66
  5144.8  187.32  5199.1  189.64  5306.4  189.96  5383.9  189.12    5615  191.25
#Mann= 4 ,-1 , 0
  4580.7     .16       0  4874.1     .07       0  5045.5     .16       0
    5615      .1       0
Bank Sta=4874.1,5045.5
XS Rating Curve= 0 ,0
Exp/Cntr=0.3,0.1

Type RM Length L Ch R = 1 ,54298   ,146,146,146
BEGIN DESCRIPTION:
Mapping XS 155d4f6a
END DESCRIPTION:
XS GIS Cut Line= 4
      2293508.43     13187031.34      2293627.21     13186875.05
      2293895.96      13186531.3      2294002.12      13186181.6
#Sta/Elev= 30
  4600.5  194.91  4668.2  192.33    4689  190.34  4774.3  185.49  4798.8  185.02
  4809.7  183.47  4845.3  181.73  4959.5  179.02  4981.5  176.07    5002  173.67
  5016.7  175.65  5037.5  175.13  5045.7  179.59  5087.3  180.85  5159.6  186.03
  5194.9  187.55  5269.1  187.71  5287.8  186.42  5300.5  186.44  5320.7  187.64
  5325.9   186.8  5342.3  188.12  5373.6   188.4  5391.7  187.81  5396.9  188.34
  5415.4  186.94  5436.3  187.04  5457.3  188.28  5488.6   188.2  5598.6  190.69
#Mann= 4 ,-1 , 0
  4600.5     .16       0  4981.5     .07       0  5037.5     .16       0
  5598.6      .1       0
Bank Sta=4959.5,5045.7
XS Rating Curve= 0 ,0
Exp/Cntr=0.3,0.1

Type RM Length L Ch R = 1 ,54152   ,408,408,408
BEGIN DESCRIPTION:
PENITAS CREEK 93.0
END DESCRIPTION:
XS GIS Cut Line= 3
      2293627.23     13187156.27      2293977.21      13186631.3
      2294077.21     13186187.56
#Sta/Elev= 30
  4540.1  197.37  4661.9  192.03  4719.7  187.71    4749   186.9    4764  184.98
  4821.1  181.18  4923.3  178.88  4972.1  180.11  4980.4  179.08  4992.4  171.33
  4995.1  170.83  5008.1  173.52  5016.4  173.11  5022.4  175.95  5044.2  179.49
  5073.5  178.86  5109.6  181.38  5124.6  183.54  5145.6  184.47  5160.6  186.46
  5166.7  185.91  5193.5  187.27  5376.8  183.77  5425.1  184.78  5431.9  185.86
  5511.6  188.82  5516.8  187.85  5565.1   189.9  5595.9  188.96  5625.9  190.54
#Mann= 4 ,-1 , 0
  4540.1     .16       0  4980.4     .07       0  5044.2     .16       0
  5625.9     .08       0
#XS Ineff= 1 ,-1
    4810 4968.75  180.11
Permanent Ineff=
       T
Bank Sta=4972.1,5044.2
XS Rating Curve= 0 ,0
Exp/Cntr=0.3,0.1

Type RM Length L Ch R = 1 ,53744   ,614,614,614
BEGIN DESCRIPTION:
PENITAS CREEK 92.0
END DESCRIPTION:
XS GIS Cut Line= 4
      2294095.95     13187500.08      2294233.46     13187175.05
      2294339.71      13186318.8      2294227.22     13185943.85
#Sta/Elev= 30
  4358.9  196.14  4377.5  195.86  4401.2  193.37  4430.3   192.5    4454  193.42
    4547  188.88  4659.8  186.15  4666.4  184.05  4683.5  186.15  4730.2  185.76
  4750.3  187.18  4786.3  183.53  4791.3  184.57  4901.5  176.98  4948.1  175.99
  4961.9  177.61    4972  177.12  4982.1  171.37  4991.9  169.58  5022.4  176.57
  5042.5  177.83  5153.4  179.01  5395.2  177.82  5633.9  185.12  5681.1  188.47
  5738.3  190.32  5804.5  190.02  5837.5  192.31  5858.6  190.87  5966.1  191.93
#Mann= 4 ,-1 , 0
  4358.9     .16       0    4972     .07       0  5042.5     .16       0
  5966.1      .1       0
#XS Ineff= 1 ,-1
 5154.64 5468.04  179.04
Permanent Ineff=
       T
Bank Sta=4961.9,5042.5
XS Rating Curve= 0 ,0
Exp/Cntr=0.3,0.1

Type RM Length L Ch R = 1 ,53130   ,1349,1349,1349
BEGIN DESCRIPTION:
PENITAS CREEK 91.0
END DESCRIPTION:
XS GIS Cut Line= 4
      2294914.71     13187493.84      2294902.21      13187281.3
      2294552.21     13186100.05      2294289.73     13185856.33
#Sta/Elev= 30
  4573.5  190.95  4653.2  188.65  4843.2  185.81  4856.9  183.29  4884.9  182.62
  4890.2  180.29  4937.1  175.47  4956.7  174.27  4961.9  179.39 4972.73  176.49
  4978.8  174.02  5000.1  169.95  5010.1  174.49  5061.6  174.11  5114.4  175.86
  5171.8  174.11  5218.7  175.91    5396  176.07  5420.1  178.14    5469  176.26
    5688  176.82  5781.9  179.56  5873.2  185.22  5906.4  185.37  5990.5  189.66
  6115.9  191.14  6122.8  189.53  6158.4  191.66  6186.8  189.99  6376.6  192.11
#Mann= 5 ,-1 , 0
  4573.5     .05       0  4653.2     .16       0 4972.73     .07       0
  5114.4     .16       0  6376.6      .1       0
#XS Ineff= 4 ,-1
 4903.27  4961.8  179.38 5139.29 5344.64  176.15 5344.64 5432.14   176.8
 5432.14 5764.29   178.1
Permanent Ineff=
       T       T       T       T
Bank Sta=4972.73,5114.4
XS Rating Curve= 0 ,0
Exp/Cntr=0.3,0.1

Type RM Length L Ch R = 1 ,51781   ,323,323,323
BEGIN DESCRIPTION:
PENITAS CREEK 90.0
END DESCRIPTION:
XS GIS Cut Line= 4
       2295064.7     13187568.82      2295214.71      13187131.3
      2295358.46      13186593.8      2295377.17     13185820.33
#Sta/Elev= 30
  4074.3  194.45  4213.8  189.49  4266.7  186.56  4456.9  183.69  4520.4   181.2
  4536.5  179.51  4665.6  175.93    4852  176.07  4945.1  173.76  4965.8  174.32
  4976.2  173.46  4986.5  168.81  4992.6  163.71  4997.6   162.4  5000.8   162.9
  5007.2  167.48  5017.6  168.64  5027.5  171.23  5032.7  171.29  5038.3  173.64
  5093.2   175.7  5160.2  174.14  5380.2  173.49  5410.2  175.02  5530.3  177.58
  5630.3  181.76  5800.4  186.52  5850.4  188.87  5860.4  188.25  5866.9  189.46
#Mann= 4 ,-1 , 0
  4074.3     .16       0  4965.8     .07       0  5038.3     .16       0
  5866.9     .08       0
#XS Ineff= 2 ,-1
 4594.64 4810.71  176.23 5089.29 5523.21  175.73
Permanent Ineff=
       T       T
Bank Sta=4976.2,5038.3
XS Rating Curve= 0 ,0
Exp/Cntr=0.3,0.1

Type RM Length L Ch R = 1 ,51458   ,698,698,698
BEGIN DESCRIPTION:
PENITAS CREEK 89.0
END DESCRIPTION:
XS GIS Cut Line= 3
      2295302.21     13187587.56      2295545.96      13187043.8
       2295852.2     13186043.83
#Sta/Elev= 30
  4059.7  193.33  4236.7  185.54  4358.1  182.25  4554.5  173.77  4600.9  173.15
    4624  170.85  4630.3  173.17  4655.6  171.01  4673.3  173.21  4814.9  176.15
  4956.4  171.36  4989.2  166.33  4994.5  162.44  4997.3  161.94  5000.5  162.44
    5008  166.66 5013.52  171.74  5021.9  172.62  5120.2  172.12  5143.9     171
    5153  167.85  5164.9   167.7    5191  169.29  5196.2  171.25  5217.2  173.32
  5321.7  177.76  5327.2  179.15  5447.2  182.13  5677.3  194.08  5701.4  194.34
#Mann= 4 ,-1 , 0
  4059.7     .16       0  4956.4     .07       0  5021.9     .16       0
  5701.4      .1       0
#XS Ineff= 2 ,-1
 4388.93 4816.43     176 5070.36 5263.21  173.05
Permanent Ineff=
       T       T
Bank Sta=4956.4,5013.52
XS Rating Curve= 0 ,0
Exp/Cntr=0.3,0.1

Type RM Length L Ch R = 1 ,50760   ,470,470,470
BEGIN DESCRIPTION:
PENITAS CREEK 88.0
END DESCRIPTION:
XS GIS Cut Line= 4
       2295339.7     13187731.31      2295758.46     13187225.05
      2296108.46      13186831.3       2296220.7     13186450.94
#Sta/Elev= 30
  4104.3  197.67  4269.1  191.37    4277  189.42  4411.1  183.71  4525.4  181.12
  4538.7  182.11  4546.6  180.88  4589.6  180.14  4688.6  180.76  4763.4  179.44
  4958.1   171.2  4964.8  170.72  4972.4  168.25  4986.3  165.85  4993.3   161.5
  4999.7  160.99  5014.2  166.06  5021.7  166.81  5028.4  164.45  5056.8  168.09
  5064.3  167.25    5071  169.37  5078.6  168.03  5120.4  169.33  5148.8  173.41
  5170.5  173.99  5184.8  175.97  5264.9  176.91  5339.1  176.82  5684.7  186.46
#Mann= 4 ,-1 , 0
  4104.3     .16       0  4972.4     .07       0  5078.6     .16       0
  5264.9      .1       0
Bank Sta=4972.4,5071
XS Rating Curve= 0 ,0
Exp/Cntr=0.3,0.1

Type RM Length L Ch R = 1 ,50290   ,566,566,566
BEGIN DESCRIPTION:
PENITAS CREEK 87.0
END DESCRIPTION:
XS GIS Cut Line= 3
       2295437.7     13187946.87      2296087.72     13187446.85
      2296887.73     13186946.85
#Sta/Elev= 30
  4199.5  201.53  4385.3  194.27    4514  186.77  4549.3  183.36  4655.3  179.33
  4719.6  174.72    4813  171.38    4919  170.22  4941.7  165.24    4948  170.03
  4969.1  168.64    4977  168.09  4983.3  166.64  4991.5  161.54  5005.8  159.25
  5012.3   160.6  5016.4  165.39  5042.6  164.67  5063.8  168.61  5121.6  173.57
  5142.8  173.23  5179.4  176.13  5432.3  178.68  5541.4  181.29  5556.7  183.34
  5585.6  182.23  5672.3  184.63    5680  186.06  5833.3  188.53    5963  193.38
#Mann= 4 ,-1 , 0
  4199.5     .16       0    4977     .07       0  5063.8     .16       0
    5963      .1       0
#XS Ineff= 1 ,-1
    4900 4948.21     170
Permanent Ineff=
       T
Bank Sta=4969.1,5063.8
XS Rating Curve= 0 ,0
Exp/Cntr=0.3,0.1

Type RM Length L Ch R = 1 ,49724   ,561,561,561
BEGIN DESCRIPTION:
PENITAS CREEK 86.0
END DESCRIPTION:
XS GIS Cut Line= 3
      2295937.76     13188146.83      2296287.72     13187946.85
      2297087.69     13187296.88
#Sta/Elev= 30
  4600.5  193.21  4769.6  181.11  4775.4  175.87  4784.7  178.21    4797   177.4
    4807  176.68  4812.8  174.04  4828.6  173.73  4842.3  171.25  4865.4  171.45
  4887.7  168.07  4909.3  166.77    4915  166.43  4974.1  164.15  4989.9  162.53
  4995.4  160.65  5017.2  161.95  5025.1  164.06  5053.9  166.73  5181.7  170.34
    5316  176.32  5423.1  177.44  5451.8  176.53  5571.7  178.07    5594   179.8
  5629.2  179.02  5736.3  182.72  5750.6  181.86  5757.1  183.09  6034.3  191.49
#Mann= 4 ,-1 , 0
  4600.5     .16       0    4915     .07       0  5053.9     .16       0
  6034.3      .1       0
Bank Sta=4909.3,5053.9
XS Rating Curve= 0 ,0
Exp/Cntr=0.3,0.1

Type RM Length L Ch R = 1 ,49163   ,551,551,551
BEGIN DESCRIPTION:
PENITAS CREEK 85.0
END DESCRIPTION:
XS GIS Cut Line= 3
      2296087.72     13188396.86      2296587.72     13188346.85
      2297337.68     13187796.88
#Sta/Elev= 30
    4492  190.23  4622.7  183.14  4713.1  176.05  4763.3  175.03  4803.5  170.77
  4934.2  166.97  4941.7  165.78  4946.8  165.37  4984.4  161.98    4989   158.6
  4991.7   158.1  5037.3  160.16  5044.1  162.04  5081.3   161.9  5102.2  162.98
  5130.9     166    5167  170.34  5208.7  172.66    5238  171.81  5329.9  172.15
  5480.4  174.27  5509.7  176.05    5539  175.63  5651.7  179.02  5660.2  180.07
    5681  179.53  5701.9  181.89  5716.6  181.18  5852.4  188.45  5924.5  192.16
#Mann= 4 ,-1 , 0
    4492     .16       0  4946.8     .07       0  5130.9     .16       0
  5852.4      .1       0
Bank Sta=4941.7,5130.9
XS Rating Curve= 0 ,0
Exp/Cntr=0.3,0.1

Type RM Length L Ch R = 1 ,48612   ,956,956,956
BEGIN DESCRIPTION:
PENITAS CREEK 84.0
END DESCRIPTION:
XS GIS Cut Line= 3
      2296387.71     13189096.86      2296837.72     13188796.85
       2297337.7     13187996.89
#Sta/Elev= 30
  4491.5  189.48  4520.1     188  4527.6   186.5  4599.7  184.47  4700.3  178.02
  4730.4  177.73  4859.6  170.19  4895.6  166.37  4910.7   166.4  4937.7  163.22
  4952.7  159.27  4973.8  159.11  5003.6  156.66  5029.3  161.56  5061.2  162.87
  5067.7  163.58    5244  168.27    5323  167.39  5396.1  168.37  5569.5  174.93
  5598.4  174.63  5692.7  178.88  5721.6  178.67  5773.5  180.43  5794.7  179.42
  5800.6  180.78    5846  181.54  5852.5  182.97  5873.7  182.19  5975.7  186.96
#Mann= 4 ,-1 , 0
  4491.5     .16       0  4937.7     .07       0  5061.2     .16       0
  5975.7     .16       0
Bank Sta=4937.7,5067.7
XS Rating Curve= 0 ,0
Exp/Cntr=0.3,0.1

Type RM Length L Ch R = 1 ,47656   ,212,212,212
BEGIN DESCRIPTION:
PENITAS CREEK 83.0
END DESCRIPTION:
XS GIS Cut Line= 3
      2296569.46     13189544.05      2297444.48     13189231.54
      2298131.98     13188825.29
#Sta/Elev= 30
  3953.1  192.02  3988.9  188.87  4068.1  186.08  4121.1  181.27    4238  174.92
  4342.5  165.64  4378.6  165.36  4434.9  162.04    4558  161.13  4630.8  162.63
  4788.5  158.01  4902.4  158.77  4923.8  157.48  4945.2     154  4982.3  156.02
  4990.5  155.09  5003.5  150.93  5013.6  154.72  5019.4  156.23 5021.35  159.71
  5025.4  169.57    5035   175.9  5040.9  171.99  5048.6  179.01  5077.9  181.18
  5099.4  180.93  5120.8  181.99  5136.5  184.48  5339.3  191.71  5680.8  200.69
#Mann= 3 ,-1 , 0
  3953.1     .16       0  4902.4     .07       0  5013.6     .16       0
#XS Ineff= 1 ,-1
 4373.21 4632.14  162.64
Permanent Ineff=
       T
Bank Sta=4902.4,5021.35
XS Rating Curve= 0 ,0
Exp/Cntr=0.3,0.1
