HEC-RAS study UNT001 IN PECR.prj: UNT001 IN PECR Base Level Engineering

--- UNT001 IN PECR.g01 (geometry) --- (continued)

Type RM Length L Ch R = 1 ,61394   ,466,466,466
BEGIN DESCRIPTION:
UNT001 IN PECR 112.0
END DESCRIPTION:
XS GIS Cut Line= 4
      2265847.27     13254132.44      2265573.84     13253845.99
      2264727.48     13253129.85      2264454.06     13252973.61
#Sta/Elev= 30
  4301.3  269.12  4354.4  265.98  4446.5  262.31  4467.6  260.42  4495.9  259.72
  4659.2  250.34  4878.1  238.03  4956.1  231.69  4998.7  227.36  5013.2  228.68
  5062.7   228.9  5134.1  230.68  5140.7  231.25  5142.4  231.25  5282.4  234.24
  5425.3  235.81  5530.7  238.11    5567  238.01  5665.8  240.86  5808.7  246.84
  5903.2  252.48  5946.4  255.97  6021.2  256.65  6042.8  259.58  6048.6  256.72
  6058.7  257.42  6070.6  261.89  6080.2  263.82  6093.6  263.03  6120.9   264.7
#Mann= 5 ,-1 , 0
  4301.3     .05       0  4659.2      .1       0  4956.1     .05       0
  5134.1      .1       0  5142.4     .05       0
Bank Sta=4956.1,5140.7
XS Rating Curve= 0 ,0
Exp/Cntr=0.3,0.1

Type RM Length L Ch R = 1 ,60928   ,549,549,549
BEGIN DESCRIPTION:
UNT001 IN PECR 111.0
END DESCRIPTION:
XS GIS Cut Line= 3
      2265837.71     13253796.83      2265537.72     13253246.85
      2265037.72     13252646.85
#Sta/Elev= 30
  4352.4  256.13  4360.4  255.06  4375.2  254.71  4463.9  248.87  4523.2  245.91
  4535.1  244.43  4573.1  242.86  4580.2  241.98  4682.7  236.74  4692.7  236.88
    4744  234.56    4808  233.34  4853.6  231.63  4899.1  229.06  4965.1  227.71
  4970.8  226.49  4989.5  225.44  4992.3  224.94  4995.5  225.44  5035.5  227.91
  5113.6  230.07  5163.1  232.18  5269.8  233.44  5323.9  233.39  5405.2  236.18
  5525.6  242.96  5553.6  243.98  5681.8  251.38  5695.5  252.62  5759.9  255.73
#Mann= 5 ,-1 , 0
  4352.4     .05       0    4744      .1       0  4989.5     .07       0
  4995.5      .1       0  5323.9     .05       0
Bank Sta=4965.1,5035.5
XS Rating Curve= 0 ,0
Exp/Cntr=0.3,0.1

Type RM Length L Ch R = 1 ,60379   ,409,409,409
BEGIN DESCRIPTION:
UNT001 IN PECR 110.0
END DESCRIPTION:
XS GIS Cut Line= 3
       2266019.1     13253820.32      2266106.51     13253053.65
      2265237.74     13252296.87
#Sta/Elev= 30
  3980.6  256.58    4125  249.95  4150.4  249.56  4165.3  249.81  4184.7  248.06
    4300  243.52  4356.5  243.01  4381.7  241.72  4631.9  236.47  4756.1  231.12
  4841.6  229.93  4911.8  226.29  4968.8  226.41  5000.9  223.15  5003.7  222.65
  5006.9  223.15    5040   224.8  5054.2  226.77  5075.1  228.52  5111.2  229.78
  5160.6  231.01  5249.3  230.62  5387.2  231.71  5476.6  234.06  5570.9  238.52
  5649.5  243.19  5691.6  246.66  5741.6   249.9  5809.6  256.05  5904.4  262.75
#Mann= 12 ,-1 , 0
  3980.6     .05       0  4150.4      .1       0    4300     .05       0
  4381.7      .1       0  5000.9     .07       0  5006.9      .1       0
  5111.2     .05       0  5249.3      .1       0  5476.6     .05       0
  5570.9      .1       0  5691.6     .08       0  5809.6     .05       0
Bank Sta=4968.8,5054.2
XS Rating Curve= 0 ,0
Exp/Cntr=0.3,0.1

Type RM Length L Ch R = 1 ,59970   ,515,515,515
BEGIN DESCRIPTION:
UNT001 IN PECR 109.0
END DESCRIPTION:
XS GIS Cut Line= 3
      2266787.75     13253246.88      2266159.72     13252648.43
      2265425.32     13252002.58
#Sta/Elev= 30
  4341.5  266.89  4394.1   263.7  4490.4  257.36    4526  254.36  4638.2  246.33
    4766     238  4843.7  231.19  4921.7  226.93  4996.4   222.4  4999.1   221.9
  5002.4   222.4  5013.5  222.41  5020.4  223.99  5034.6  224.83  5098.5  226.87
  5119.5  229.09  5134.3  229.39    5304  230.67  5482.6  229.72  5629.5   230.5
  5657.9  232.26  5664.6  234.05  5693.1  236.59  5813.6  239.08  5835.4  238.49
    5888  240.85  6005.2  248.73  6054.5  250.55  6062.1  252.05    6187  254.81
#Mann= 10 ,-1 , 0
  4341.5      .1       0  4394.1     .05       0  4490.4      .1       0
    4526     .05       0  4638.2      .1       0  4996.4     .07       0
  5002.4      .1       0  5134.3     .05       0  5482.6      .1       0
    5888     .05       0
Bank Sta=4921.7,5098.5
XS Rating Curve= 0 ,0
Exp/Cntr=0.3,0.1

Type RM Length L Ch R = 1 ,59455   ,481,481,481
BEGIN DESCRIPTION:
UNT001 IN PECR 108.0
END DESCRIPTION:
XS GIS Cut Line= 3
      2266964.57     13253140.74      2266773.27     13252773.23
      2266557.05     13251299.93
#Sta/Elev= 30
    4328  267.68  4439.9  263.79  4674.5  245.86  4737.5  240.61  4749.9  240.21
  4758.9  238.97  4789.2   237.5  4819.8  234.27  4859.9  231.66  4890.3  228.48
  4940.8  225.57  4954.3  223.55  4998.4  221.33  5001.2  220.83  5004.4  221.33
  5011.5  222.24  5041.9  223.45  5072.2  223.46  5112.6  225.39  5142.9  226.19
  5193.5  224.96  5228.5  226.99  5284.4  226.86  5457.7  228.75  5587.7  230.42
  5769.6  230.41  5870.7  234.48  6062.7  245.35  6120.9  249.65  6231.4  254.81
#Mann= 5 ,-1 , 0
    4328     .05       0  4674.5      .1       0  4998.4     .07       0
  5004.4      .1       0  5457.7     .05       0
Bank Sta=4940.8,5112.6
XS Rating Curve= 0 ,0
Exp/Cntr=0.3,0.1

Type RM Length L Ch R = 1 ,58974   ,341,341,341
BEGIN DESCRIPTION:
UNT001 IN PECR 107.0
END DESCRIPTION:
XS GIS Cut Line= 4
      2267181.06     13252596.97      2267095.49     13252400.66
      2266813.54     13251554.83      2266768.57     13251309.96
#Sta/Elev= 30
  4499.7  253.08  4541.8  252.64  4570.7  250.49  4576.2  248.92  4587.1  248.49
  4608.9  245.59    4623  245.13  4675.3  239.92  4723.8  237.42  4786.1  233.56
  4833.8  229.31  4844.1   229.2  4854.9   226.9  4918.1  223.35    4939   223.6
  4944.2  222.75  4970.6  222.18  4975.9  220.12  4988.9  219.47  4991.7  218.97
  4994.9  219.47  5102.3  224.02  5234.9  226.98  5508.2  229.21  5571.4  231.97
  5694.9  239.12  5766.1  245.02  5778.7  246.95  5837.2  251.21  5854.4  251.71
#Mann= 5 ,-1 , 0
  4499.7     .05       0  4723.8      .1       0  4988.9     .07       0
  4994.9      .1       0  5234.9     .05       0
Bank Sta=4939,5102.3
XS Rating Curve= 0 ,0
Exp/Cntr=0.3,0.1

Type RM Length L Ch R = 1 ,58633   ,278,278,278
BEGIN DESCRIPTION:
UNT001 IN PECR 106.0
END DESCRIPTION:
XS GIS Cut Line= 4
      2267322.05     13252481.23      2267347.22     13252143.89
      2267055.21     13251413.86      2266899.15      13251126.9
#Sta/Elev= 30
    4391  251.01  4405.4  250.92  4435.5   248.6  4511.7  244.53  4545.8  243.04
  4585.9  239.93  4706.3  234.07  4782.6  230.37  4887.6  223.45  4927.6   221.9
    4963  222.07  4981.5  220.88  4995.3  218.58  5002.7  218.13  5005.4  217.63
  5008.7  218.13  5016.9   219.5  5059.5  221.77  5139.8  224.37  5189.2  225.53
    5310  226.63  5441.9  231.01  5584.8  240.23  5591.8  241.37  5710.2     248
  5739.8  250.59  5748.2  250.55  5797.6  253.64  5829.9  254.31  5842.2  255.41
#Mann= 7 ,-1 , 0
    4391     .05       0  4511.7      .1       0  4706.3     .05       0
  4782.6      .1       0  5002.7     .07       0  5008.7      .1       0
  5139.8     .05       0
Bank Sta=4963,5059.5
XS Rating Curve= 0 ,0
Exp/Cntr=0.3,0.1

Type RM Length L Ch R = 1 ,58355   ,548,548,548
BEGIN DESCRIPTION:
UNT001 IN PECR 105.0
END DESCRIPTION:
XS GIS Cut Line= 4
       2267503.3     13252435.92      2267568.75     13252103.61
       2267372.4     13251293.02      2267055.67     13250991.38
#Sta/Elev= 30
    4292  249.02  4343.9  247.17  4423.5  242.25  4441.5  240.45  4550.3  234.54
  4654.7  228.97  4689.1  228.26  4696.5  227.28  4738.3  225.72  4905.2  221.33
  4952.5  221.34  4962.3  220.65  4987.5  218.81  4996.5  217.13  4999.3  216.63
  5002.5  217.13  5036.2  220.73  5069.8  222.01  5090.4  222.99  5147.7  223.49
  5255.6   225.1  5297.4  227.06  5429.9  235.49  5459.5  236.52  5472.2  237.84
  5592.7  243.94    5628  244.59  5691.8  247.29  5790.6   249.3  5902.1  254.01
#Mann= 6 ,-1 , 0
    4292      .1       0  4550.3     .05       0  4962.3      .1       0
  4996.5     .07       0  5002.5      .1       0  5147.7     .05       0
Bank Sta=4952.5,5069.8
XS Rating Curve= 0 ,0
Exp/Cntr=0.3,0.1

Type RM Length L Ch R = 1 ,57807   ,92,92,92
BEGIN DESCRIPTION:
Mapping XS 5d56d4dd
END DESCRIPTION:
XS GIS Cut Line= 4
       2267956.6     13252596.37      2268055.56     13251622.39
      2267935.76     13251507.81      2267873.38     13250930.73
#Sta/Elev= 30
  3941.4  248.26  4004.1  245.34  4041.4  242.06  4192.2  236.52  4197.6  235.56
    4353  232.29    4544  223.56  4865.6  221.66  4936.9  219.97  4944.1  218.46
  4948.6   215.9    4951  214.54  4979.4  209.24  5011.6  207.84  5014.3  207.34
  5017.6  207.84    5057  215.46  5064.3  218.98  5071.2  219.92  5089.2  219.95
  5113.4  221.88  5296.9  224.41  5348.6  226.65  5429.1  231.45  5459.3  234.55
  5509.6   236.7  5577.3  243.68  5582.3  243.28  5640.3  247.88  5666.6  251.25
#Mann= 5 ,-1 , 0
  3941.4      .1       0  4197.6     .05       0  4948.6      .1       0
  5011.6     .07       0  5017.6      .1       0
Bank Sta=4936.9,5071.2
XS Rating Curve= 0 ,0
Exp/Cntr=0.3,0.1

Type RM Length L Ch R = 1 ,57715   ,157,157,157
BEGIN DESCRIPTION:
UNT001 IN PECR 104.0
END DESCRIPTION:
XS GIS Cut Line= 4
      2268029.52     13252580.71      2268149.31     13251585.93
      2268008.68     13251455.73      2267967.01     13250903.61
#Sta/Elev= 30
  3894.6  249.51  4079.8  239.26  4150.3  236.89  4168.9     235  4452.5  227.83
  4512.9  225.89  4589.5  221.83  4815.1  221.86  4875.2  220.17  4875.7  220.17
  4899.6  221.85  4904.1  223.44  4911.4  223.37  4918.2  224.71  4925.6  224.23
  4932.4  225.94  4946.6  224.73  5031.6  224.43    5060  224.58  5066.8  226.03
  5088.2  225.77  5097.1  227.24  5107.1  226.99  5137.2  223.33  5164.9  222.09
  5287.6  225.02  5458.1  236.56  5548.4  244.42  5578.5  247.93  5641.9  251.61
#Mann= 3 ,-1 , 0
  3894.6      .1       0  4875.7     .05       0  5066.8      .1       0
#XS Ineff= 2 , 0
       0 4918.33  224.72  5099.8       0  227.25
Permanent Ineff=
       T       T
Bank Sta=4932.4,5066.8
XS Rating Curve= 0 ,0
Exp/Cntr=0.3,0.1

Type RM Length L Ch R = 1 ,57558   ,690,690,690
BEGIN DESCRIPTION:
UNT001 IN PECR 103.0
END DESCRIPTION:
XS GIS Cut Line= 4
      2268087.72     13252596.88      2268258.68     13251518.23
      2268138.89     13251346.35      2268092.05     13250841.54
#Sta/Elev= 30
  3824.3   251.3  4006.6  240.31  4101.4  236.33  4174.6  232.51  4279.9  229.68
  4441.9  228.74  4496.3  226.92  4558.7  223.25    4621  221.59  4755.8  220.96
  4846.9  221.49  4904.2  220.23  4920.3     220  4925.5  219.29  4954.7  219.07
  5003.2   215.6  5006.4   216.1  5032.8  218.98  5047.7  219.08  5053.8  220.83
  5062.5   220.4  5068.6  222.35  5076.5  220.47  5089.5  220.64  5245.9  225.53
  5376.5  233.27  5410.4  234.15  5416.7  235.33  5446.8  237.72  5632.9  249.06
#Mann= 5 ,-1 , 0
  3824.3      .1       0  4101.4     .05       0  4904.2      .1       0
  4920.3     .05       0  5006.4      .1       0
Bank Sta=4920.3,5053.8
XS Rating Curve= 0 ,0
Exp/Cntr=0.3,0.1

Type RM Length L Ch R = 1 ,56868   ,704,704,704
BEGIN DESCRIPTION:
UNT001 IN PECR 102.0
END DESCRIPTION:
XS GIS Cut Line= 3
      2268987.72      13252596.9      2268887.72     13251396.85
      2268837.71     13251046.81
#Sta/Elev= 30
  3795.4  245.71  4046.3  235.92  4076.4  234.31    4099  232.25  4126.6  232.18
    4142  230.94  4146.7  230.28  4176.8  229.79  4206.9  228.24  4219.4  228.36
  4226.9  227.52  4297.2  224.36  4417.6  220.83  4575.6  220.18  4580.7  220.66
  4638.4  219.41  4701.1  219.57  4788.9  217.36  4849.1  218.82  4899.3  216.97
  4921.6  217.47  4959.5  217.12  4989.3  213.38  5019.8  216.02  5029.9  217.35
  5080.4  220.27    5242  231.79  5302.6  234.71  5352.2  238.95  5353.2  238.95
#Mann= 6 ,-1 , 0
  3795.4      .1       0    4142     .05       0  4921.6      .1       0
  4959.5     .05       0  5019.8      .1       0  5352.2     .05       0
Bank Sta=4959.5,5029.9
XS Rating Curve= 0 ,0
Exp/Cntr=0.3,0.1

Type RM Length L Ch R = 1 ,56164   ,491,491,491
BEGIN DESCRIPTION:
UNT001 IN PECR 101.0
END DESCRIPTION:
XS GIS Cut Line= 3
      2269592.01     13252466.14      2269459.74     13251527.81
      2268887.72     13250946.86
#Sta/Elev= 30
  4052.4  243.76  4265.5  234.11  4314.2  230.76  4400.8     227  4455.6  225.14
  4545.1  220.48  4588.1  219.77  4623.3  219.18  4687.5  218.41    4900  218.33
  4930.3  216.06  4970.7  212.86  4977.2  212.99  4987.9  211.48  4990.6  210.98
  4993.9  211.48  5004.2  211.99  5016.2   213.7  5058.6  216.31  5126.2  217.05
  5221.3  216.18  5299.1  216.48  5405.2  220.58  5419.3  220.28  5617.4  231.33
  5624.4   232.3  5695.1  236.44  5709.2   238.2  5751.7  239.94  5815.3  244.06
#Mann= 7 ,-1 , 0
  4052.4     .05       0  4400.8      .1       0  4588.1     .05       0
  4623.3      .1       0  4987.9     .07       0  4993.9      .1       0
  5126.2     .05       0
Bank Sta=4930.3,5058.6
XS Rating Curve= 0 ,0
Exp/Cntr=0.3,0.1

Type RM Length L Ch R = 1 ,55673   ,343,343,343
BEGIN DESCRIPTION:
UNT001 IN PECR 100.0
END DESCRIPTION:
XS GIS Cut Line= 3
      2270037.71     13252646.81      2269837.72     13251246.85
      2269887.72     13250446.88
#Sta/Elev= 30
  3573.9  254.56  3695.1  251.22  3836.5  245.65  3876.9  242.52  3907.2  241.21
  3917.3  239.86  4028.4  233.46  4114.5  227.13  4210.2  221.47  4270.9  218.87
  4301.2     219  4341.6  217.36  4553.7     217  4634.5  218.34  4712.8  217.44
  4856.7  216.46    4887   214.7  4947.7  213.85    4978  211.77  5005.1  210.98
  5007.9  210.48  5011.1  210.98  5038.2  213.53  5138.4  215.67  5268.6   223.2
  5378.8  228.12  5499.1  236.39  5551.7  238.51  5559.2  239.62  5789.6  252.04
#Mann= 5 ,-1 , 0
  3573.9      .1       0  4114.5     .05       0  4712.8      .1       0
  5005.1     .07       0  5011.1      .1       0
Bank Sta=4947.7,5038.2
XS Rating Curve= 0 ,0
Exp/Cntr=0.3,0.1

Type RM Length L Ch R = 1 ,55330   ,789,789,789
BEGIN DESCRIPTION:
UNT001 IN PECR 99.0
END DESCRIPTION:
XS GIS Cut Line= 3
       2270276.3     13252428.56      2270261.54     13251933.86
      2270084.52     13250510.35
#Sta/Elev= 30
  3712.1  247.18  3773.8  245.11  3911.9  236.93    4104  225.81    4274  218.35
  4375.3   216.3  4481.8  215.51  4617.2  215.29    4673   215.5  4840.6  216.14
  4925.6  212.63  4949.7  212.66  4969.9  214.43  4979.9  214.02    4990  209.05
  4997.1  206.97  4999.8  206.47  5003.1  206.97  5006.5  208.66  5040.4  211.89
  5050.5  214.76  5060.6  215.32  5070.6  214.22  5092.3  214.22  5161.3  219.76
    5254  224.79  5292.3  227.96  5403.2  232.37  5433.4  234.79  5641.5  245.56
#Mann= 8 ,-1 , 0
  3712.1      .1       0  3911.9     .05       0  4481.8      .1       0
  4617.2     .05       0    4673     .16       0  4840.6      .1       0
  4997.1     .07       0  5003.1      .1       0
Bank Sta=4979.9,5050.5
XS Rating Curve= 0 ,0
Exp/Cntr=0.3,0.1

Type RM Length L Ch R = 1 ,54541   ,533,533,533
BEGIN DESCRIPTION:
UNT001 IN PECR 98.0
END DESCRIPTION:
XS GIS Cut Line= 3
      2270519.97     13252295.65      2270652.87     13251668.04
      2271132.56     13250531.55
#Sta/Elev= 30
    3645  240.27  4103.7  223.24  4239.6   220.4  4360.8  219.33  4524.8   213.3
  4566.8  211.45  4619.7  210.91  4737.8  213.48    4761  213.34  4854.8  213.61
  4902.2  211.21  4931.3  210.84  4971.6  211.95  4984.2  208.97  4993.3  205.81
  5002.5  205.66  5004.9  204.58  5007.7  204.08  5010.9  204.58  5015.1  207.56
  5025.9  211.24  5084.5  212.53  5108.2  215.68  5177.9  221.61  5208.5  226.03
    5285  232.41  5297.3  234.15  5396.2  241.74    5491  246.14  5520.1  248.55
#Mann= 6 ,-1 , 0
    3645     .05       0  4524.8      .1       0  4737.8     .16       0
    4761      .1       0  5004.9     .07       0  5010.9      .1       0
Bank Sta=4971.6,5025.9
XS Rating Curve= 0 ,0
Exp/Cntr=0.3,0.1

Type RM Length L Ch R = 1 ,54008   ,709,709,709
BEGIN DESCRIPTION:
UNT001 IN PECR 97.0
END DESCRIPTION:
XS GIS Cut Line= 3
      2270787.74     13252496.82      2271337.72     13251246.85
      2271537.71     13250896.87
#Sta/Elev= 30
  3649.5   245.2  3739.3  243.79  3811.7  240.83    3868  238.63  4082.5  225.88
  4195.7   220.5  4310.4   216.7  4416.9  215.45  4512.7  214.38  4643.7  208.52
  4826.4  212.11  4904.4  210.81  4925.2  211.11  4960.5  208.32  4971.4  208.62
  4977.4  210.15  4993.3  207.54  4997.7  204.05  5000.5  203.55  5003.7  204.05
  5012.4  206.25    5018  206.25    5023   209.5  5044.6  209.25  5103.6   212.1
  5153.3  217.46    5175  218.43  5202.3  221.63  5286.5  229.91  5418.2  239.02
#Mann= 10 ,-1 , 0
  3649.5      .1       0  3811.7     .05       0  4310.4      .1       0
  4416.9     .16       0  4512.7      .1       0  4904.4     .12       0
  4997.7     .07       0  5003.7     .12       0    5175      .1       0
  5202.3     .05       0
Bank Sta=4977.4,5023
XS Rating Curve= 0 ,0
Exp/Cntr=0.3,0.1

Type RM Length L Ch R = 1 ,53299   ,479,479,479
BEGIN DESCRIPTION:
UNT001 IN PECR 96.0
END DESCRIPTION:
XS GIS Cut Line= 4
      2271029.41     13252502.43      2271310.02     13252199.67
      2271701.35     13251601.59       2271767.8     13251276.74
#Sta/Elev= 30
  4287.8  246.29  4306.9  245.26  4361.5  242.49    4446  236.49  4460.2  234.55
  4559.4  226.62  4723.5  216.55  4810.3  212.61  4852.5  210.02    4946  207.13
  4976.2  207.02  4982.1  207.77  4990.8  202.93  5000.2  201.22    5003  200.72
  5006.2  201.22  5012.4  201.36  5026.6  206.26  5033.4  205.98  5039.4  207.78
  5048.5  207.64  5054.5  208.62  5111.8  207.81  5178.2  209.52  5256.6  213.66
  5271.7  215.09  5562.8  223.98  5625.6  225.95    5676  228.46  5746.9  229.94
#Mann= 6 ,-1 , 0
  4287.8      .1       0  4306.9     .05       0  4723.5      .1       0
  5000.2     .07       0  5006.2      .1       0  5562.8     .05       0
Bank Sta=4982.1,5026.6
XS Rating Curve= 0 ,0
Exp/Cntr=0.3,0.1

Type RM Length L Ch R = 1 ,52820   ,443,443,443
BEGIN DESCRIPTION:
UNT001 IN PECR 95.0
END DESCRIPTION:
XS GIS Cut Line= 4
      2271406.03     13252805.12       2271723.5     13252620.54
       2271952.4     13251815.72       2271952.4     13251359.89
#Sta/Elev= 30
  4251.8  236.55  4456.7   222.5  4521.3  218.74  4552.7  217.97  4558.5   217.1
  4622.8  214.42  4689.9  212.24  4851.6  209.73  4976.3  204.72  4981.6  202.26
  4994.1   198.9  4996.9   198.4  5000.1   198.9  5007.5   203.2  5015.5  205.03
  5020.7  203.45  5028.3  205.74  5044.1  205.77  5145.9  207.16  5224.9  209.35
    5251  209.06  5371.4  211.71  5419.3  214.16  5451.4  214.15  5474.6  214.18
  5550.3  216.56  5644.6  219.19  5704.6  222.06  5804.6  225.15  5911.6  227.45
#Mann= 10 ,-1 , 0
  4251.8     .05       0  4622.8      .1       0  4994.1     .07       0
  5000.1      .1       0  5044.1     .16       0  5145.9     .05       0
  5224.9      .1       0    5251     .05       0  5451.4      .1       0
  5550.3     .05       0
Bank Sta=4976.3,5015.5
XS Rating Curve= 0 ,0
Exp/Cntr=0.3,0.1

Type RM Length L Ch R = 1 ,52377   ,468,468,468
BEGIN DESCRIPTION:
UNT001 IN PECR 94.0
END DESCRIPTION:
XS GIS Cut Line= 4
       2272904.9     13253152.17      2272543.09     13252775.59
       2272269.9     13252487.63      2272159.14     13251372.68
#Sta/Elev= 30
  3919.2   243.2    4027  238.86  4229.3  226.67  4370.3  217.92  4430.1  213.74
  4550.3  208.85  4628.3  207.33  4691.8  203.55  4727.4   203.9  4790.9  206.85
    4814   206.6  4881.5  205.82  4969.8  203.99  4989.9  200.78  4996.9  197.63
  4999.7  197.13  5002.9  197.63  5013.6  198.91    5020  203.41  5040.1  204.85
  5114.4  205.63  5170.8  208.57  5233.3  208.92    5311  208.56  5532.5   211.1
  5719.3  219.93  5793.8  221.61  5825.2  224.74  5904.4  226.84  5958.8  226.87
#Mann= 8 ,-1 , 0
  3919.2      .1       0  4229.3     .05       0  4370.3      .1       0
    4814     .16       0  4881.5      .1       0  4996.9     .07       0
  5002.9      .1       0  5233.3     .05       0
Bank Sta=4969.8,5020
XS Rating Curve= 0 ,0
Exp/Cntr=0.3,0.1

Type RM Length L Ch R = 1 ,51909   ,605,605,605
BEGIN DESCRIPTION:
UNT001 IN PECR 93.0
END DESCRIPTION:
XS GIS Cut Line= 2
      2272937.72     13252846.84      2272380.74     13251530.96
#Sta/Elev= 30
  4421.7   231.7  4443.6  230.26    4541  225.55  4606.3  221.53  4612.9  220.25
  4689.4   214.4    4780   209.1  4842.4  206.01  4918.9  204.34  4971.7   201.9
  4975.5  202.41  4977.1  202.62  4986.3  201.26  4997.8  196.49  5000.5  195.99
  5003.8  196.49  5024.5  203.29  5111.6  204.29  5124.6  203.95  5277.6  206.87
  5456.3  206.91  5527.7  206.88    5589  207.33  5659.6  210.77  5670.9  212.16
  5789.3   217.4  5800.8  218.53  5825.3  219.19  5833.3  219.29  5850.6  221.17
#Mann= 10 ,-1 , 0
  4421.7      .1       0  4443.6     .05       0    4541      .1       0
  4975.5     .16       0  4997.8     .07       0  5003.8     .16       0
  5111.6      .1       0  5456.3     .05       0  5527.7      .1       0
  5825.3     .05       0
Bank Sta=4977.1,5024.5
XS Rating Curve= 0 ,0
Exp/Cntr=0.3,0.1

Type RM Length L Ch R = 1 ,51304   ,464,464,464
BEGIN DESCRIPTION:
UNT001 IN PECR 92.0
END DESCRIPTION:
XS GIS Cut Line= 3
      2273637.76     13252246.87      2273237.72     13252046.85
      2272437.68     13251446.83
#Sta/Elev= 30
  4542.5  222.39  4628.3  217.95  4796.9  209.78  4819.3  210.11  4891.9  202.73
  4908.7   202.4  4914.3  200.81  4931.1  201.59  4936.6   200.3  4953.4  203.39
    4959  199.81  4961.5  200.37  4968.3  201.48  4981.4  198.87    4987  196.18
    4994  195.66  4996.8  195.16    5000  195.66  5003.3  195.78  5017.9  201.35
  5078.4  202.18  5145.5  202.38  5226.2  205.32  5326.2  207.07  5532.5  205.57
  5661.2  206.86  5772.5  212.22  5772.8  212.24  5918.8  220.02  5989.8  223.54
#Mann= 12 ,-1 , 0
  4542.5      .1       0  4628.3     .05       0  4961.5     .16       0
  4968.3     .05       0    4994     .04       0    5000     .05       0
  5078.4      .1       0  5145.5     .05       0  5661.2      .1       0
  5772.5     .05       0  5772.8      .1       0  5918.8     .05       0
Bank Sta=4968.3,5017.9
XS Rating Curve= 0 ,0
Exp/Cntr=0.3,0.1

Type RM Length L Ch R = 1 ,50840   ,507,507,507
BEGIN DESCRIPTION:
UNT001 IN PECR 91.0
END DESCRIPTION:
XS GIS Cut Line= 3
      2273987.73     13252146.87      2273537.72     13251696.85
      2272737.71     13251046.85
#Sta/Elev= 30
  4331.7  232.51    4558  218.66  4652.3  214.52  4812.6  207.49  4859.9  204.54
  4939.8  199.43  4968.1  199.19  4981.7  198.44  4989.7  193.75  4993.1  192.79
  4995.9  192.29  4999.1  192.79  5024.9  201.06  5109.8  200.96  5175.4   203.9
  5202.3   204.9  5266.2  205.14  5309.3  204.38  5373.2  205.53  5422.8  205.48
  5480.3  204.13    5565  204.89  5586.6  204.34  5636.9  205.31  5771.2  209.52
  5814.3  212.84  5913.4  218.28  5921.3  219.64  5970.7  222.37  5998.9  223.25
#Mann= 7 ,-1 , 0
  4331.7      .1       0  4652.3     .05       0  4859.9      .1       0
  4993.1     .07       0  4999.1      .1       0  5175.4     .05       0
  5970.7      .1       0
Bank Sta=4968.1,5024.9
XS Rating Curve= 0 ,0
Exp/Cntr=0.3,0.1

Type RM Length L Ch R = 1 ,50333   ,526,526,526
BEGIN DESCRIPTION:
UNT001 IN PECR 90.0
END DESCRIPTION:
XS GIS Cut Line= 3
      2274387.75     13251946.88      2273887.72     13251346.85
      2273087.69     13250846.83
#Sta/Elev= 30
  4211.6  239.53  4467.4  224.48  4473.9  224.79  4481.7  223.61  4701.7  210.11
  4737.3  208.98  4824.8  205.03  4893.1  202.25  4928.2  199.75  4971.2  199.51
    4979  198.59  4985.5  196.27  4989.4  193.31  4995.6  193.31  4997.3  191.98
  5000.1  191.48  5003.3  191.98  5015.7  198.93  5021.6  199.94  5051.6  200.67
  5122.4  199.16  5185.7  203.54  5236.9   203.7    5268  202.68  5350.6  203.56
  5566.4  204.84  5681.9  209.94  5733.8     211  5834.1  215.65  5936.1  218.73
#Mann= 8 ,-1 , 0
  4211.6      .1       0  4737.3     .05       0  4824.8      .1       0
  4997.3     .07       0  5003.3      .1       0  5185.7     .05       0
  5236.9      .1       0  5350.6     .05       0
Bank Sta=4971.2,5015.7
XS Rating Curve= 0 ,0
Exp/Cntr=0.3,0.1

Type RM Length L Ch R = 1 ,49807   ,575,575,575
BEGIN DESCRIPTION:
UNT001 IN PECR 89.0
END DESCRIPTION:
XS GIS Cut Line= 3
      2274687.71     13251746.84      2274237.72     13250946.85
       2273637.7     13250146.83
#Sta/Elev= 30
  4117.6  239.03  4184.8  236.88  4255.6  232.65  4346.7  225.14  4427.4  220.77
  4433.4  219.16  4476.8   217.4    4552  211.49  4655.4  205.38  4800.6  199.83
  4816.5  200.29  4924.9  197.74  4958.2  199.23  4978.1  199.07  4989.9  193.02
  5002.8  190.39  5005.6  189.89  5008.8  190.39  5012.5  193.47  5021.8  193.26
  5027.5  195.26  5038.6  195.35  5042.8  197.81  5071.9  198.07  5171.9   200.9
  5307.3  201.68  5471.9  205.16  5673.6  214.66  5963.6  232.46  6035.5   235.8
#Mann= 7 ,-1 , 0
  4117.6      .1       0  4655.4     .05       0  4958.2      .1       0
  5002.8     .07       0  5008.8      .1       0  5071.9     .05       0
  5673.6      .1       0
Bank Sta=4978.1,5042.8
XS Rating Curve= 0 ,0
Exp/Cntr=0.3,0.1

Type RM Length L Ch R = 1 ,49232   ,399,399,399
BEGIN DESCRIPTION:
UNT001 IN PECR 88.0
END DESCRIPTION:
XS GIS Cut Line= 3
      2274861.57     13251623.76       2274802.5     13251239.79
       2274713.9     13250331.68
#Sta/Elev= 30
  4312.4   236.8  4441.1  231.91    4461  229.84  4491.4  224.85  4562.2  219.72
  4567.6  217.78  4612.8  215.74  4630.8  213.31  4693.7  208.58  4699.1   207.2
  4723.9  205.26  4800.4  200.14  4842.2  198.47  4932.6  196.16  4965.1     196
  4985.2  193.32  4995.2   189.2  5003.9  191.25  5005.9  188.89  5008.7  188.39
  5011.9  188.89  5015.3  192.88  5025.4  196.47  5035.4  197.32  5055.5  196.42
  5110.6  196.66  5171.4  198.43  5286.6  202.47  5467.4  211.25  5613.3  213.71
#Mann= 6 ,-1 , 0
  4312.4      .1       0  4842.2     .05       0  4932.6      .1       0
  5005.9     .07       0  5011.9      .1       0  5171.4     .05       0
Bank Sta=4965.1,5025.4
XS Rating Curve= 0 ,0
Exp/Cntr=0.3,0.1

Type RM Length L Ch R = 1 ,48833   ,369,369,369
BEGIN DESCRIPTION:
UNT001 IN PECR 87.0
END DESCRIPTION:
XS GIS Cut Line= 3
      2275238.13     13251328.35      2275230.75     13251121.65
      2274862.15     13250325.47
#Sta/Elev= 30
  4613.9  231.55  4645.4  232.61  4665.4  231.14  4685.4  228.09  4735.5  222.65
  4745.5  220.02    4768  218.02  4795.5  213.68  4864.1   208.1  4870.1  206.85
  4961.3  197.44  4978.7  194.41  4984.2  195.03  4991.3  187.31  4998.6  186.09
  5001.4  185.59  5004.6  186.09  5013.4  194.47  5024.4  195.87  5167.6  195.11
  5207.7  195.74  5255.7  196.98  5287.7  197.54    5366  202.77  5460.5  208.05
  5498.2  208.82  5520.3   210.6  5567.6  212.29  5663.5  215.15  5698.1   215.4
#Mann= 8 ,-1 , 0
  4613.9      .1       0  4998.6     .07       0  5004.6      .1       0
  5207.7     .05       0  5255.7      .1       0    5366     .05       0
  5460.5      .1       0  5567.6     .05       0
Bank Sta=4984.2,5013.4
XS Rating Curve= 0 ,0
Exp/Cntr=0.3,0.1

Type RM Length L Ch R = 1 ,48464   ,678,678,678
BEGIN DESCRIPTION:
UNT001 IN PECR 86.0
END DESCRIPTION:
XS GIS Cut Line= 3
      2275548.25     13251055.21      2275563.02     13250870.61
       2274994.5     13250206.11
#Sta/Elev= 30
  4609.7  217.98  4658.2  218.22  4669.5  216.96  4708.4  215.95  4758.5  213.08
  4787.4  209.66  4829.4  207.19  4837.1  205.38  4872.2  201.55  4878.8  200.12
  4893.1  199.45    4915  196.84  4943.6  194.47  4968.1  194.37  4978.7  194.68
  4996.6  185.07  4999.3  184.57  5002.6  185.07  5013.8  193.63  5028.1  194.92
  5042.4  193.35  5070.9  193.21  5097.2  194.49  5101.5  194.73  5234.1  197.41
  5552.8  210.15  5581.4  210.71  5609.9  209.74  5630.8  210.49  5669.4     210
#Mann= 6 ,-1 , 0
  4609.7      .1       0  4968.1     .12       0  4996.6     .07       0
  5002.6     .12       0  5097.2      .1       0  5101.5     .05       0
Bank Sta=4978.7,5013.8
XS Rating Curve= 0 ,0
Exp/Cntr=0.3,0.1

Type RM Length L Ch R = 1 ,47786   ,410,410,410
BEGIN DESCRIPTION:
UNT001 IN PECR 85.0
END DESCRIPTION:
XS GIS Cut Line= 3
       2275654.5     13250997.42      2276047.43     13250422.39
      2275393.01     13249565.96
#Sta/Elev= 30
  4070.9  213.91    4282  210.15  4398.5   209.6  4404.6  208.65  4470.3  209.33
  4476.4  208.16  4664.7  205.83  4762.1  202.94  4785.4  202.93  4806.7  202.35
  4856.8  199.87  4935.7  192.31  4972.8  193.16  4977.4  193.28  4985.6  190.86
  4991.9  182.15  4997.1  181.52  4999.9  181.02  5003.1  181.52  5013.4  188.64
    5021  192.43  5027.2  193.64  5058.5  192.06    5100   192.5    5312  197.48
  5498.9  206.48    5542  206.46  5563.3  209.52  5750.8  218.68  5845.2   223.1
#Mann= 11 ,-1 , 0
  4070.9      .1       0  4762.1     .16       0  4785.4      .1       0
  4806.7     .16       0  4972.8     .12       0  4997.1     .07       0
  5003.1     .12       0  5058.5     .16       0    5100      .1       0
    5312     .05       0  5750.8      .1       0
Bank Sta=4972.8,5021
XS Rating Curve= 0 ,0
Exp/Cntr=0.3,0.1

Type RM Length L Ch R = 1 ,47376   ,662,662,662
BEGIN DESCRIPTION:
UNT001 IN PECR 84.0
END DESCRIPTION:
XS GIS Cut Line= 3
      2276508.13     13250634.35      2276367.84     13250220.84
      2275769.74     13249334.77
#Sta/Elev= 30
  4205.6  213.28  4652.3  198.88  4745.2  194.51  4754.1  195.82  4803.9  195.16
  4826.1  193.45  4832.1  191.29    4862  194.08  4943.6   191.9    4970  192.01
    4976  186.18    4988  182.88  4990.7  182.38    4994  182.88  5005.9  183.28
    5012  188.97  5026.9  191.72  5041.9  191.33  5056.9  185.27  5065.2  185.91
  5069.3  185.54  5092.8  191.42  5158.9  194.08  5242.8  199.61  5308.7  198.48
  5452.6  203.19  5489.6   206.6  5639.7  212.33  5673.4  214.13  5711.3   215.7
#Mann= 9 ,-1 , 0
  4205.6      .1       0  4943.6     .12       0    4988     .07       0
    4994     .12       0  5065.2     .12       0  5158.9      .1       0
  5489.6     .08       0  5639.7      .1       0  5673.4     .08       0
Bank Sta=4970,5026.9
XS Rating Curve= 0 ,0
Exp/Cntr=0.3,0.1

Type RM Length L Ch R = 1 ,46714   ,509,509,509
BEGIN DESCRIPTION:
UNT001 IN PECR 83.0
END DESCRIPTION:
XS GIS Cut Line= 3
      2276663.18     13250604.84      2276663.18     13250272.53
      2276677.95     13249157.63
#Sta/Elev= 30
  3971.8  211.47  4149.8  206.79  4249.8  200.66  4329.8   197.3  4479.5  194.89
  4491.6  194.59  4594.1  194.11  4614.2  194.16  4779.8  192.87  4879.8  189.52
  4959.8  191.86  4979.8  190.39 4981.25  189.36  4996.8  178.02  4999.6  177.52
  5002.8  178.02  5009.8  179.85  5019.6   187.1 5026.25  187.78  5029.8  190.48
  5199.9  209.84  5229.9   214.6  5249.9  216.75  5259.9  216.52  5269.9  219.38
  5279.9  219.68  5299.9  223.18  5349.9  224.87  5359.9  227.95  5419.1  233.61
#Mann= 7 ,-1 , 0
  3971.8      .1       0  4479.5     .08       0  4491.6      .1       0
  4594.1     .16       0  4614.2      .1       0  4996.8     .07       0
  5002.8      .1       0
Bank Sta=4981.25,5026.25
XS Rating Curve= 0 ,0
Exp/Cntr=0.3,0.1

Type RM Length L Ch R = 1 ,46205   ,533,533,533
BEGIN DESCRIPTION:
UNT001 IN PECR 82.0
END DESCRIPTION:
XS GIS Cut Line= 4
      2276818.25     13250730.29      2276951.15     13250434.97
      2277202.19     13249504.63      2277135.74     13249283.14
#Sta/Elev= 30
  3935.5  210.98  4072.3  205.05  4158.6  203.48  4170.4  202.12  4211.2  203.32
    4307   199.7  4408.5  195.56  4458.3  193.45  4567.7  192.34  4868.5  191.26
  4881.8  190.81  4916.5  186.49  4921.7  187.84  4951.2  181.96  4956.4  182.69
  4982.4  181.06  4991.1  182.43  4993.3  180.59  4996.1  180.09  4999.3  180.59
  5036.2  181.76  5044.6   184.3  5054.9  185.41  5065.3  189.44    5071  191.89
  5076.1  190.63  5150.8  198.29  5256.5  206.08  5304.2  210.83  5454.2   220.1
#Mann= 5 ,-1 , 0
  3935.5      .1       0    4307     .08       0  4408.5      .1       0
  4993.3     .07       0  4999.3      .1       0
Bank Sta=4921.7,5065.3
XS Rating Curve= 0 ,0
Exp/Cntr=0.3,0.1

Type RM Length L Ch R = 1 ,45672   ,527,527,527
BEGIN DESCRIPTION:
UNT001 IN PECR 81.0
END DESCRIPTION:
XS GIS Cut Line= 3
      2277128.48     13250872.38       2277706.6     13249783.85
      2277487.83     13249356.74
#Sta/Elev= 30
  3985.4  212.43  4012.2  212.36  4025.6  209.71  4070.9   207.8  4100.1  204.51
  4144.1  203.27  4172.8  200.11  4195.5  198.48  4204.4  199.12  4218.1  197.31
  4263.4  195.58  4408.6  194.08  4424.7  193.88    4693  192.81  4818.2  188.61
  4863.2  188.88  4912.8  186.45  4973.1  186.15  4978.8     182  4992.1  176.76
  4994.8  176.26  4998.1  176.76  5010.7  178.35  5017.1  187.03  5022.7  187.99
  5067.3  186.91  5356.5  200.38  5511.9  202.58  5607.8  206.97  5697.8  209.43
#Mann= 5 ,-1 , 0
  3985.4      .1       0  4408.6     .08       0  4424.7      .1       0
  4992.1     .07       0  4998.1      .1       0
Bank Sta=4973.1,5017.1
XS Rating Curve= 0 ,0
Exp/Cntr=0.3,0.1

Type RM Length L Ch R = 1 ,45145   ,510,510,510
BEGIN DESCRIPTION:
UNT001 IN PECR 80.0
END DESCRIPTION:
XS GIS Cut Line= 2
      2278287.74     13250496.89      2277550.36     13249263.04
#Sta/Elev= 30
    4591  214.12  4684.4  208.84  4707.5  208.19  4765.8  203.14  4801.1  201.49
  4838.1  197.72  4917.9  191.64    4949  188.06  4963.8  187.74  4970.4   186.3
  4976.2  184.48    4986  178.74  4991.8  177.35  4995.8  174.43  4998.5  173.93
  5001.8  174.43  5007.4  177.31  5022.1  181.23  5028.8  186.09  5138.6  185.72
  5209.7  186.37    5342  189.48    5379  191.27  5421.8  191.84  5575.4  199.63
  5639.6  201.55  5802.6  201.89  5931.5  205.83  5962.6  205.91  6028.4  207.85
#Mann= 3 ,-1 , 0
    4591      .1       0  4995.8     .07       0  5001.8      .1       0
Bank Sta=4970.4,5028.8
XS Rating Curve= 0 ,0
Exp/Cntr=0.3,0.1

Type RM Length L Ch R = 1 ,44635   ,546,546,546
BEGIN DESCRIPTION:
UNT001 IN PECR 79.0
END DESCRIPTION:
XS GIS Cut Line= 3
      2278587.72     13250296.86      2278487.72     13249846.85
       2277687.7     13249096.83
#Sta/Elev= 30
  4547.5  218.93  4571.8   217.3  4578.2  215.07    4609  213.37  4615.4  211.72
  4799.8  198.75  4916.3   186.5  4957.3  184.89  4967.5  181.86  4977.7  183.81
  4984.1  181.87  4989.3  175.25  4995.2  173.69    4998  173.19  5001.2  173.69
  5011.9  174.97  5015.6  178.89  5022.4  183.27  5029.7  184.74  5072.2  183.52
  5277.4  188.36  5482.5  197.63  5517.7  201.32  5560.2  198.01  5581.7  197.85
  5588.5  196.34    5610  196.47  5616.9  194.66  5694.5     194  6105.1  210.26
#Mann= 3 ,-1 , 0
  4547.5      .1       0  4995.2     .07       0  5001.2      .1       0
Bank Sta=4977.7,5022.4
XS Rating Curve= 0 ,0
Exp/Cntr=0.3,0.1

Type RM Length L Ch R = 1 ,44089   ,637,637,637
BEGIN DESCRIPTION:
UNT001 IN PECR 78.0
END DESCRIPTION:
XS GIS Cut Line= 3
      2279254.86     13249962.42      2278538.64     13249032.07
      2278486.97     13248441.63
#Sta/Elev= 30
  4391.3  213.42  4414.2  213.53  4499.4  208.68  4600.2  201.06  4613.5  198.42
  4650.7  197.84  4727.7  192.26  4885.4  187.38  4978.7  182.74  4985.1  179.36
  4991.5  172.99  4996.6  171.51  4999.3  171.01  5002.6  171.51  5020.4  181.88
  5034.9  182.98  5049.4  181.35  5178.1  185.08  5256.5  185.43  5306.7  188.88
  5377.4  191.73  5412.7  194.64  5441.7   195.2  5462.5  197.29    5671  206.16
  5731.3  205.66  5747.2  203.41  5761.4  205.42  5901.9  205.88  6158.1  214.58
#Mann= 3 ,-1 , 0
  4391.3      .1       0  4996.6     .07       0  5002.6      .1       0
Bank Sta=4978.7,5020.4
XS Rating Curve= 0 ,0
Exp/Cntr=0.3,0.1

Type RM Length L Ch R = 1 ,43452   ,480,480,480
BEGIN DESCRIPTION:
UNT001 IN PECR 77.0
END DESCRIPTION:
XS GIS Cut Line= 3
      2279572.35     13249740.92      2279476.36     13249393.87
      2278967.72     13248450.31
#Sta/Elev= 30
  4141.9  212.67  4180.2  212.01  4248.9  209.38  4288.4  206.92  4301.7  207.01
  4367.4  202.78  4488.5  197.35    4502  197.54  4556.4  193.81  4588.9  193.34
  4594.5  192.18  4676.5  188.39  4771.2   185.4  4807.8  185.79  4862.1  184.02
    4906  181.29  4941.6  181.84  4977.3  181.04  4993.6  173.52  4996.2  171.57
    4999  171.07  5002.2  171.57  5021.2  181.05  5103.1  182.42  5214.3  191.47
  5288.8  196.53  5407.4  200.63  5436.4  202.72    5524  205.18  5573.9  208.38
#Mann= 3 ,-1 , 0
  4141.9      .1       0  4996.2     .07       0  5002.2      .1       0
Bank Sta=4977.3,5021.2
XS Rating Curve= 0 ,0
Exp/Cntr=0.3,0.1

Type RM Length L Ch R = 1 ,42972   ,533,533,533
BEGIN DESCRIPTION:
UNT001 IN PECR 76.0
END DESCRIPTION:
XS GIS Cut Line= 3
      2279787.71     13249496.82      2279637.72     13248696.85
      2279237.71     13248296.85
#Sta/Elev= 30
  4185.6  207.86  4195.7  206.76  4205.9  206.96  4211.8  205.91  4256.8  204.26
    4317  200.59  4348.4   199.7  4427.2  194.82  4531.5  190.68  4623.1   188.1
  4647.6  188.72  4684.1  186.67  4700.2  187.04  4724.8  186.14  4765.5  183.43
  4973.2  178.86    4994  169.04  4996.7  168.54    5000  169.04    5003  169.04
  5027.8  178.72  5084.4  181.37  5098.5  183.48  5126.8   183.5  5140.9  179.66
  5183.4  187.28  5310.6  194.62  5367.2  196.94  5409.6  200.12  5565.2  208.79
#Mann= 3 ,-1 , 0
  4185.6      .1       0    4994     .07       0    5000      .1       0
Bank Sta=4973.2,5027.8
XS Rating Curve= 0 ,0
Exp/Cntr=0.3,0.1

Type RM Length L Ch R = 1 ,42439   ,416,416,416
BEGIN DESCRIPTION:
UNT001 IN PECR 75.0
END DESCRIPTION:
XS GIS Cut Line= 3
      2280030.14     13249519.38      2280103.97     13249128.06
      2280236.83     13247991.42
#Sta/Elev= 30
  4127.5  206.82  4195.8  203.62  4201.3  202.43  4248.2  199.53  4253.3  199.93
  4300.6  195.66  4305.7  196.06  4523.8  185.07  4708.2  182.94  4879.3  178.55
  4929.7  177.93  4959.9  179.09    4980  178.23  4990.1  172.11  5000.1  168.12
  5007.2  167.83    5010  167.33  5013.2  167.83  5020.3  174.05  5028.5  178.69
  5040.4   178.5  5050.5  180.83  5090.7  185.43  5100.8  185.55  5116.9  188.27
  5151.2   191.8  5221.6  196.64    5282  198.35  5548.7  196.64  5670.1  199.15
#Mann= 3 ,-1 , 0
  4127.5      .1       0  5007.2     .07       0  5013.2      .1       0
Bank Sta=4980,5028.5
XS Rating Curve= 0 ,0
Exp/Cntr=0.3,0.1

Type RM Length L Ch R = 1 ,42023   ,632,632,632
BEGIN DESCRIPTION:
UNT001 IN PECR 74.0
END DESCRIPTION:
XS GIS Cut Line= 4
      2280295.96     13249548.92      2280487.93     13249297.88
      2280569.15     13248493.06       2280502.7     13248005.81
#Sta/Elev= 30
  4199.3  203.79  4252.3  204.29  4365.6  201.51    4637  184.33  4687.2  181.79
  4765.8  181.14  4822.2  180.29  4968.6  176.14  4978.7  174.74  4981.8  173.19
  4995.8   166.1  4998.5   165.6  5001.8   166.1  5008.8  167.43  5018.9  173.64
  5028.9  175.88  5079.2  178.53  5109.4  182.94  5157.4  187.33  5209.9  193.53
  5280.2  198.09  5330.5  198.65  5441.1   194.8  5512.2  193.52  5523.6  194.54
  5562.6  193.05  5683.7  194.81    5714  196.53  5740.5  196.08    5816  199.94
#Mann= 7 ,-1 , 0
  4199.3      .1       0  4765.8     .12       0  4822.2      .1       0
  4981.8     .12       0  4995.8     .07       0  5001.8     .12       0
  5157.4      .1       0
Bank Sta=4968.6,5028.9
XS Rating Curve= 0 ,0
Exp/Cntr=0.3,0.1

Type RM Length L Ch R = 1 ,41391   ,592,592,592
BEGIN DESCRIPTION:
UNT001 IN PECR 73.0
END DESCRIPTION:
XS GIS Cut Line= 4
      2281441.66     13249734.88      2281176.91     13249400.69
      2281120.49     13248888.54      2280659.13     13247904.42
#Sta/Elev= 30
  4172.2  196.97  4208.5  195.15  4216.6  193.79  4222.9  191.11  4249.4  189.14
  4520.7  188.31    4603  187.13  4662.8  179.89  4704.2  178.18  4749.6  176.94
  4793.6  176.17  4833.8   177.2    4864  175.77  4954.5  175.26  4964.6  173.18
  4974.6  168.74    5003  166.58  5005.7  166.08    5009  166.58  5014.9  171.25
 5034.09  175.89    5035  177.15  5112.1  180.84  5251.8  183.44  5402.8  188.94
  5582.4  190.11  5645.3  188.48    5839  191.99  5998.7  196.35  6200.7   204.8
#Mann= 7 ,-1 , 0
  4172.2      .1       0  4249.4     .05       0  4520.7      .1       0
  4704.2     .16       0  4749.6      .1       0    5003     .07       0
    5009      .1       0
Bank Sta=4954.5,5034.09
XS Rating Curve= 0 ,0
Exp/Cntr=0.3,0.1

Type RM Length L Ch R = 1 ,40799   ,523,523,523
BEGIN DESCRIPTION:
UNT001 IN PECR 72.0
END DESCRIPTION:
XS GIS Cut Line= 2
      2281863.79     13249497.29      2281239.11     13248076.01
#Sta/Elev= 30
    4500  191.85  4621.3  191.87  4678.7  191.55  4730.8  188.31  4754.2  183.63
  4762.6  176.03  4784.5  170.51  4800.5  169.78  4829.7  171.39  4847.6  168.74
  4882.8  172.43  4923.1  174.12  4975.3  173.85  4981.1  170.49  5001.1  163.92
  5003.8  163.42  5007.1  163.92  5013.9  170.81    5022  173.69  5064.7  174.92
  5090.3  174.67    5173  178.05  5222.7  178.05    5378  179.46  5483.6  178.89
  5527.3  180.55  5606.6  180.54  5756.7  181.02  5899.3   185.7  6052.5  186.08
#Mann= 9 ,-1 , 0
    4500     .05       0  4621.3      .1       0  4800.5     .16       0
  5001.1     .07       0  5007.1     .16       0  5064.7      .1       0
  5222.7     .05       0    5378     .08       0  5606.6      .1       0
Bank Sta=4975.3,5022
XS Rating Curve= 0 ,0
Exp/Cntr=0.3,0.1

Type RM Length L Ch R = 1 ,40276   ,976,976,976
BEGIN DESCRIPTION:
UNT001 IN PECR 71.0
END DESCRIPTION:
XS GIS Cut Line= 2
      2282259.97     13249242.75      2281765.16     13247513.55
#Sta/Elev= 30
  4660.2  191.45  4801.5   192.7  4811.9  190.63  4834.9  179.06  4843.1  170.41
  4874.4  166.38    4916   168.3  4926.4  171.63  4957.6  172.81    4968  171.94
  4988.8  167.07  4996.2  161.19  4998.9  160.69  5002.2  161.19  5014.2  164.61
    5020  169.36  5030.4  170.95    5048  173.68  5186.4  172.49  5285.5  174.72
  5363.2  176.51  5827.4  174.73  5848.3  174.61  5862.5  176.04  5887.3  175.04
  5954.8  175.88  6027.6  177.91  6091.3  182.09  6164.1  184.16  6458.8   198.8
#Mann= 5 ,-1 , 0
  4660.2      .1       0  4996.2     .07       0  5002.2      .1       0
  5285.5     .05       0  5827.4      .1       0
Bank Sta=4968,5030.4
XS Rating Curve= 0 ,0
Exp/Cntr=0.3,0.1

Type RM Length L Ch R = 1 ,39300   ,1165,1165,1165
BEGIN DESCRIPTION:
Mapping XS cd1abceb
END DESCRIPTION:
XS GIS Cut Line= 4
      2282442.27     13249065.59      2282890.16     13248518.75
      2282593.29     13247935.41      2282884.96     13247294.78
#Sta/Elev= 30
  3999.2  192.28    4045  193.26  4142.2  190.15  4223.7  184.75  4242.2  183.59
  4336.8  178.05  4442.7  174.78    4663  174.51  4863.2  171.26  4962.5  169.61
  4977.5   166.8  4990.7  161.07  5004.3  159.76  5007.1  159.26  5010.3  159.76
  5012.9  165.48  5029.6  169.49  5067.2  169.76  5089.7  166.81  5115.5  170.24
  5171.9  173.62  5185.3  174.99  5213.1  173.61  5402.7  173.93  5481.3  172.64
  5633.7  173.57  5798.8  187.15  5831.5  188.13  5897.4  195.26  6064.5  205.15
#Mann= 13 ,-1 , 0
  3999.2      .1       0  4142.2     .05       0  4223.7      .1       0
  4242.2     .05       0  4336.8      .1       0  4863.2     .16       0
  4962.5     .12       0  5004.3     .07       0  5010.3     .12       0
  5115.5     .16       0  5171.9      .1       0  5402.7     .05       0
  5481.3      .1       0
Bank Sta=4962.5,5029.6
XS Rating Curve= 0 ,0
Exp/Cntr=0.3,0.1

Type RM Length L Ch R = 1 ,38135   ,344,344,344
BEGIN DESCRIPTION:
UNT001 IN PECR 70.0
END DESCRIPTION:
XS GIS Cut Line= 3
      2282509.96     13249107.28      2283739.12      13248112.5
      2283525.78     13247701.43
#Sta/Elev= 30
  3672.1  189.96    3762  189.83  3812.5  187.73  3876.8  182.58  3891.4  181.85
  3999.3  176.34  4196.7  172.69  4645.1  172.63  4851.7  171.47    4930  167.51
  4957.2  161.59  4965.2  163.49  4971.6  160.63  4974.7  161.35  4979.6  162.49
    4986   159.7  5004.1  158.62  5006.9  158.12  5010.1  158.62  5014.8  158.95
  5029.1  164.72  5035.6  163.64  5064.3  166.75  5227.4  182.58  5393.4  186.08
  5406.2  188.94  5481.9   194.9  5592.5   197.7  5598.1  199.19  5716.5  200.54
#Mann= 9 ,-1 , 0
  3672.1      .1       0    3762     .05       0  3876.8      .1       0
  3891.4     .05       0  3999.3      .1       0  4645.1     .05       0
  4974.7      .1       0  5004.1     .07       0  5010.1      .1       0
Bank Sta=4930,5064.3
XS Rating Curve= 0 ,0
Exp/Cntr=0.3,0.1

Type RM Length L Ch R = 1 ,37791   ,644,644,644
BEGIN DESCRIPTION:
UNT001 IN PECR 69.0
END DESCRIPTION:
XS GIS Cut Line= 2
      2283082.86     13249461.47       2283968.6     13248235.09
#Sta/Elev= 30
  3832.3  187.89  3861.4  187.29  3911.7  183.05  3947.2   181.8  3961.4  179.73
  4008.5  177.26  4104.3  173.63  4133.7  173.85  4169.3  171.94    4341  170.78
  4441.6  169.02  4541.1  169.61  4613.3  171.36  4849.5  170.68  4948.3  165.37
  4971.5  165.45  4977.7  161.87  4985.2  160.21  4992.4  155.46  4995.6  155.33
  4998.3  154.83  5001.6  155.33    5028  160.86  5042.7   165.6  5084.5  167.07
  5120.9   171.4  5157.9  174.49  5170.3  176.52  5264.7  182.43  5345.1  185.77
#Mann= 4 ,-1 , 0
  3832.3     .05       0  4008.5      .1       0  4995.6     .07       0
  5001.6      .1       0
Bank Sta=4971.5,5042.7
XS Rating Curve= 0 ,0
Exp/Cntr=0.3,0.1

Type RM Length L Ch R = 1 ,37147   ,461,461,461
BEGIN DESCRIPTION:
UNT001 IN PECR 68.0
END DESCRIPTION:
XS GIS Cut Line= 3
      2284287.72     13249696.84      2284244.69     13249008.31
      2284228.75     13248379.99
#Sta/Elev= 30
  4236.9  200.14  4266.9  198.82    4287  196.34  4301.7  193.56  4367.1  185.21
  4413.8  182.74  4467.3  179.66  4479.9  179.51  4517.4  176.77  4635.2  171.02
  4868.1  164.81  4889.6  165.11  4918.2  164.66  4938.2  163.61  4968.2  163.49
  4988.3  156.24  4995.3  155.53    4998  155.03  5001.3  155.53  5008.8  155.59
  5018.3  159.08  5028.3  161.52  5038.3  162.69  5128.3  164.67  5221.3  169.85
  5288.3  174.26  5401.1  178.79  5458.4  181.89  5518.4  183.47  5555.3  183.45
#Mann= 7 ,-1 , 0
  4236.9      .1       0  4301.7     .08       0  4413.8     .05       0
  4889.6      .1       0  4995.3     .07       0  5001.3      .1       0
  5221.3     .05       0
Bank Sta=4968.2,5038.3
XS Rating Curve= 0 ,0
Exp/Cntr=0.3,0.1

Type RM Length L Ch R = 1 ,36686   ,601,601,601
BEGIN DESCRIPTION:
UNT001 IN PECR 67.0
END DESCRIPTION:
XS GIS Cut Line= 4
      2284740.22     13249740.03      2284774.95     13249375.45
      2284549.25     13248490.04       2284306.8     13248351.49
#Sta/Elev= 30
  4193.9  191.93  4317.6  182.07  4324.2  180.65  4448.2   173.5  4518.5   170.8
  4641.2  168.74  4867.1  167.36  4934.4  166.05  4940.5  164.62  4961.1  162.67
  4970.1  159.12  4992.1  154.34  4999.4  153.84  5002.2  153.34  5005.4  153.84
  5016.2  157.07  5023.1   157.9  5033.4  160.72  5043.7  162.07  5064.3  163.15
  5126.3  163.26  5143.9  164.06  5215.4  166.27  5302.4  165.86  5384.3  170.54
  5491.6  170.53  5579.3     174  5625.3  177.23  5690.3  180.05  5753.1  181.25
#Mann= 5 ,-1 , 0
  4193.9     .05       0  4867.1      .1       0  4999.4     .07       0
  5005.4      .1       0  5143.9     .05       0
Bank Sta=4961.1,5043.7
XS Rating Curve= 0 ,0
Exp/Cntr=0.3,0.1

Type RM Length L Ch R = 1 ,36085   ,895,895,895
BEGIN DESCRIPTION:
UNT001 IN PECR 66.0
END DESCRIPTION:
XS GIS Cut Line= 3
      2285387.72     13249396.84      2285137.72     13248596.85
       2284587.7     13247796.82
#Sta/Elev= 30
  4202.1   188.9  4296.4  184.59    4335  181.56  4423.7  176.39  4579.3  171.41
  4663.1  166.88    4904  163.41  4921.3   161.2  4937.7  159.21  4945.9  158.67
    4959  154.45  4986.3  153.34  4995.3  151.28  4998.1  150.78  5001.3  151.28
  5018.8  154.92    5024  160.85  5076.6  160.95  5123.9  163.49  5161.6  165.53
  5298.7  167.62  5415.1  164.51  5513.8  165.38  5537.5  164.47  5615.3  166.23
  5672.7   165.4  5773.6  169.21  5788.5   171.1  5809.4  171.61  6011.1  186.18
#Mann= 7 ,-1 , 0
  4202.1      .1       0    4335     .05       0  4937.7      .1       0
  4995.3     .07       0  5001.3      .1       0  5123.9     .05       0
  5672.7      .1       0
Bank Sta=4921.3,5024
XS Rating Curve= 0 ,0
Exp/Cntr=0.3,0.1

Type RM Length L Ch R = 1 ,35190   ,780,780,780
BEGIN DESCRIPTION:
UNT001 IN PECR 65.0
END DESCRIPTION:
XS GIS Cut Line= 3
      2285639.53     13249292.85      2285697.86     13248276.84
      2285586.08     13247411.71
#Sta/Elev= 30
  3638.7  182.44  3724.8     178  3895.1  173.64  3975.2  174.15  4185.6  180.45
    4494  172.01  4516.1  170.76  4636.3  170.62  4676.5  172.21    4737  170.84
  4807.6  166.67    4858  161.91  4958.9  158.36    4979  156.11  4989.1  151.49
  5003.4   147.6  5006.2   147.1  5009.4   147.6  5019.4  151.26  5029.4  157.98
  5041.9  159.18    5052  159.94  5200.9  179.07  5271.4  184.31  5318.8  190.14
  5392.4  196.42  5403.2  200.17  5412.6  205.61  5452.9  208.33  5528.7  208.55
#Mann= 6 ,-1 , 0
  3638.7     .05       0    4494      .1       0  5003.4     .07       0
  5009.4      .1       0  5041.9     .12       0    5052      .1       0
Bank Sta=4958.9,5029.4
XS Rating Curve= 0 ,0
Exp/Cntr=0.3,0.1

Type RM Length L Ch R = 1 ,34410   ,350,350,350
BEGIN DESCRIPTION:
UNT001 IN PECR 64.0
END DESCRIPTION:
XS GIS Cut Line= 2
      2285756.18     13249390.07      2286582.57     13247708.12
#Sta/Elev= 30
  3774.5  188.84  4106.8  170.43  4202.3  167.29  4286.6  166.91  4292.2   165.4
    4324  168.47  4346.3  166.78  4427.1   168.5  4736.2  166.87  4825.4  163.42
  4914.6  157.05  4959.1  157.51  4972.2  156.09  4975.5  154.21  4981.4  150.84
  5000.7  147.16  5003.4  146.66  5006.7  147.16  5011.6  147.26    5026  153.39
  5039.6  154.75  5107.1  159.92    5197  173.25  5264.4  179.13  5371.3  191.21
  5399.3  196.02  5438.2  199.29  5472.3  205.76  5579.2  211.63  5648.5  213.17
#Mann= 4 ,-1 , 0
  3774.5     .05       0  4975.5      .1       0  5000.7     .07       0
  5006.7      .1       0
Bank Sta=4972.2,5039.6
XS Rating Curve= 0 ,0
Exp/Cntr=0.3,0.1
