HEC-RAS study UNT001 IN PECR.prj: UNT001 IN PECR Base Level Engineering

--- UNT001 IN PECR.g01 (geometry) --- (continued)

Type RM Length L Ch R = 1 ,34060   ,202,202,202
BEGIN DESCRIPTION:
UNT001 IN PECR 63.0
END DESCRIPTION:
XS GIS Cut Line= 2
      2285999.54     13249487.49       2286884.7     13247951.48
#Sta/Elev= 30
  3894.9   192.9  4121.1  177.62    4288  168.08    4415     164  4523.5  162.53
  4584.1  162.23  4764.7  163.97  4922.1  156.07  4978.8  154.45  4984.5  148.98
  5012.2  147.35  5014.9  146.85  5018.2  147.35  5037.7  154.33  5072.9  154.69
  5118.1  156.74  5123.9  158.55  5144.5  158.45  5176.8  157.69  5182.8  160.89
  5198.6  161.44  5204.3  160.11  5211.4  163.37  5352.4  171.62  5402.6  175.07
  5461.5   177.5  5467.3  176.64  5498.8  179.43  5504.6  178.33  5667.7  185.09
#Mann= 8 ,-1 , 0
  3894.9     .05       0  4523.5     .08       0  4584.1     .05       0
  4922.1      .1       0  5012.2     .07       0  5018.2      .1       0
  5144.5     .12       0  5352.4     .08       0
Bank Sta=4978.8,5037.7
XS Rating Curve= 0 ,0
Exp/Cntr=0.3,0.1

Type RM Length L Ch R = 1 ,33858   ,792,792,792
BEGIN DESCRIPTION:
UNT001 IN PECR 62.0
END DESCRIPTION:
XS GIS Cut Line= 2
      2286098.51      13249690.6       2287004.7     13248091.75
#Sta/Elev= 30
  3826.6  202.65  3846.1  200.38  3922.9  192.38  4029.1  185.21  4069.4  182.83
  4239.1  174.71  4342.3  171.49  4401.4  167.61  4466.3   167.6  4474.6  168.73
  4482.2  167.29    4488  168.51    4527  166.74    4825  159.96  4864.6  158.52
  4870.3   157.1    4967  155.86  4972.7   154.6  4988.6  151.39  4991.4  148.05
  4994.1  147.55  4997.4  148.05  5031.9  148.44  5047.8   154.4  5112.7  157.07
  5215.1  166.51  5302.2  172.22  5376.7  175.87  5405.7   175.9  5664.4  189.33
#Mann= 9 ,-1 , 0
  3826.6      .1       0  3846.1     .08       0  4029.1      .1       0
  4069.4     .08       0  4239.1      .1       0    4527     .08       0
    4825      .1       0  4991.4     .07       0  4997.4      .1       0
Bank Sta=4972.7,5047.8
XS Rating Curve= 0 ,0
Exp/Cntr=0.3,0.1

Type RM Length L Ch R = 1 ,33066   ,845,845,845
BEGIN DESCRIPTION:
UNT001 IN PECR 61.0
END DESCRIPTION:
XS GIS Cut Line= 2
      2286358.94     13249893.73      2287332.83     13249112.53
#Sta/Elev= 30
  4137.9  186.26    4185  183.56  4220.2  180.28  4269.8  178.32  4298.6  175.84
  4490.7  165.47  4625.1   160.7  4789.9  159.38  4903.6  153.18  4945.2  154.39
  4959.6  150.68  4967.6  147.19    4974  146.35    4982  142.73  4988.4  143.08
  4992.3  141.39    4995  140.89  4998.3  141.39  5017.2  145.58  5023.6  149.17
  5031.6  151.68  5052.4  152.03  5081.2  155.99    5102  157.37  5130.8  163.79
  5180.4     169    5230  175.66    5294  178.01  5358.1   177.9  5386.4  176.55
#Mann= 3 ,-1 , 0
  4137.9      .1       0  4992.3     .07       0  4998.3      .1       0
Bank Sta=4959.6,5031.6
XS Rating Curve= 0 ,0
Exp/Cntr=0.3,0.1

Type RM Length L Ch R = 1 ,32221   ,403,403,403
BEGIN DESCRIPTION:
UNT001 IN PECR 60.0
END DESCRIPTION:
XS GIS Cut Line= 2
      2286968.31     13250471.85      2287806.83     13249654.17
#Sta/Elev= 30
  4468.9  194.75  4493.3   194.8  4528.6  190.72  4549.9  189.83  4648.9  175.49
    4670  174.23  4691.3  170.72  4792.8  160.94  4938.8  150.25  4942.3  148.88
  4967.1  139.73    4974  141.37  4985.2  139.41  4987.9  138.91  4991.2  139.41
  5016.5   141.8  5030.6  148.46  5051.9  149.75  5066.1  148.95  5094.4  150.71
  5115.5   153.5  5122.7  152.81  5129.6   153.5  5136.8  157.07  5157.9  158.74
  5192.1  158.74  5213.7  157.98  5341.8  152.48    5455  153.44  5640.1  163.55
#Mann= 7 ,-1 , 0
  4468.9      .1       0  4792.8     .12       0  4942.3      .1       0
  4985.2     .07       0  4991.2      .1       0  5192.1     .12       0
  5213.7      .1       0
Bank Sta=4942.3,5030.6
XS Rating Curve= 0 ,0
Exp/Cntr=0.3,0.1

Type RM Length L Ch R = 1 ,31818   ,311,311,311
BEGIN DESCRIPTION:
UNT001 IN PECR 59.0
END DESCRIPTION:
XS GIS Cut Line= 3
      2287437.74     13250646.82      2287687.72     13250296.85
      2287837.71      13249696.9
#Sta/Elev= 30
  4550.9  192.68    4573  193.73  4579.1   191.6  4587.7  192.39  4629.5   190.5
    4659  194.13  4709.4  194.35  4736.4  190.78  4751.2  181.55  4772.1   173.4
  4795.4   169.3  4881.4  158.92  4931.8  149.64  4944.1  149.27  4952.7  143.22
  4970.6  138.83  4973.4  138.33  4976.6  138.83    4999  139.49  5022.2  145.59
  5032.5  146.64  5040.2  149.67  5127.9  150.79  5197.5  154.64  5228.4  154.34
  5251.6  151.52  5259.3  149.37  5317.3  151.62  5465.4  157.02  5599.4  164.09
#Mann= 5 ,-1 , 0
  4550.9      .1       0  4970.6     .07       0  4976.6      .1       0
  5197.5     .12       0  5317.3      .1       0
Bank Sta=4944.1,5040.2
XS Rating Curve= 0 ,0
Exp/Cntr=0.3,0.1

Type RM Length L Ch R = 1 ,31507   ,780,780,780
BEGIN DESCRIPTION:
UNT001 IN PECR 58.0
END DESCRIPTION:
XS GIS Cut Line= 3
      2288037.72     13250746.87      2288004.75     13250357.29
      2287900.58     13249706.25
#Sta/Elev= 30
  4515.7  172.62    4573  169.36    4578  170.08    4606  167.41  4692.5  162.73
  4736.5  161.78  4786.7  162.36  4811.9  160.04  4909.4  156.55  4937.5  149.47
  4957.8  146.86  4967.9  148.13  4977.9  145.19  4982.9  139.71  5005.4   139.2
  5008.1   138.7  5011.4   139.2  5028.6  147.26  5069.2  149.35  5089.4  146.21
    5107  148.42  5112.1  147.57    5148  150.86  5221.1   153.8  5299.8  152.83
  5360.2  152.43  5422.2  153.52  5489.3  157.34    5535  161.43    5566  162.46
#Mann= 5 ,-1 , 0
  4515.7      .1       0  5005.4     .07       0  5011.4      .1       0
    5148     .12       0  5299.8      .1       0
Bank Sta=4967.9,5028.6
XS Rating Curve= 0 ,0
Exp/Cntr=0.3,0.1

Type RM Length L Ch R = 1 ,30727   ,528,528,528
BEGIN DESCRIPTION:
UNT001 IN PECR 57.0
END DESCRIPTION:
XS GIS Cut Line= 3
      2288437.73     13250646.84      2288687.72     13249996.85
      2288837.72     13249446.84
#Sta/Elev= 30
  4329.7  170.85  4374.7  168.99  4415.4  161.35    4486  156.71  4563.2  150.95
  4668.9  148.61  4746.8  149.06  4886.8  147.93  4931.8  144.94  4951.1  146.89
    4991  134.41  4993.7  133.91    4997  134.41  5011.1   137.3  5016.5  140.59
  5028.7  139.58  5057.2  146.69  5077.9  151.38  5106.7  151.82  5143.4  154.04
  5212.7  160.78  5236.9  160.04  5385.4  173.92  5499.4  181.81  5544.4  187.98
  5565.1  188.48  5573.7  191.04  5578.9  189.59  5585.8  195.38  5596.2  199.38
#Mann= 8 ,-1 , 0
  4329.7     .05       0    4486      .1       0  4668.9     .05       0
  4746.8      .1       0    4991     .07       0    4997      .1       0
  5106.7     .16       0  5143.4      .1       0
Bank Sta=4951.1,5057.2
XS Rating Curve= 0 ,0
Exp/Cntr=0.3,0.1

Type RM Length L Ch R = 1 ,30199   ,543,543,543
BEGIN DESCRIPTION:
UNT001 IN PECR 56.0
END DESCRIPTION:
XS GIS Cut Line= 3
      2288623.51     13250909.04       2289247.1     13250118.31
      2289311.39      13249584.7
#Sta/Elev= 30
  4381.2  175.88  4613.2     166  4713.9  159.84  4842.2  147.84  4930.3  145.13
  4969.8   144.6  4976.8  143.18  4991.3  134.15  4994.6  134.06  4997.4  133.56
  5000.6  134.06  5020.1  135.45  5026.5  138.24  5047.3  143.93  5055.4  145.43
  5076.2  143.52  5105.1  147.52  5169.2  151.67  5268.6   153.9  5409.8  159.48
  5419.9  161.09  5510.6   166.3  5517.2  167.63    5571   171.2  5591.1   171.3
  5651.6  176.81  5762.4  183.46  5768.5  186.36  5773.6  184.34  5925.7   194.9
#Mann= 4 ,-1 , 0
  4381.2     .05       0  4930.3      .1       0  4994.6     .07       0
  5000.6      .1       0
Bank Sta=4969.8,5047.3
XS Rating Curve= 0 ,0
Exp/Cntr=0.3,0.1

Type RM Length L Ch R = 1 ,29656   ,646,646,646
BEGIN DESCRIPTION:
UNT001 IN PECR 55.0
END DESCRIPTION:
XS GIS Cut Line= 4
      2289047.83     13251185.43      2289272.81     13250992.59
       2289787.1     13250208.31      2289703.52     13249944.72
#Sta/Elev= 30
  4382.7  171.71  4495.1  162.56  4630.1  153.83  4721.8  150.95  4875.3  149.84
  4902.4  144.96  4932.6   142.6  4953.7  141.84  4960.9  143.28  4974.7  141.68
  4986.8  132.57  4989.6  132.07  4992.8  132.57  5003.9  133.02    5026  136.81
  5032.7  142.54  5068.5  142.03  5140.5  145.05  5164.2  149.48  5170.7  149.29
  5176.7  147.07  5191.8  146.21  5300.3  147.02  5393.7  153.92  5460.1  160.63
  5574.6   161.2  5648.8  163.94  5754.8  169.57  5786.3  172.76  5893.4  177.65
#Mann= 5 ,-1 , 0
  4382.7     .05       0  4986.8     .03       0  4992.8     .05       0
  5003.9      .1       0  5648.8     .05       0
Bank Sta=4974.7,5032.7
XS Rating Curve= 0 ,0
Exp/Cntr=0.3,0.1

Type RM Length L Ch R = 1 ,29010   ,491,491,491
BEGIN DESCRIPTION:
UNT001 IN PECR 54.0
END DESCRIPTION:
XS GIS Cut Line= 3
      2290153.52     13251461.85      2289999.24     13250446.16
      2289877.08     13250156.83
#Sta/Elev= 30
  4417.7  168.87  4519.2   169.4  4591.1  167.24  4655.4  161.67  4707.2  156.13
  4838.7  146.06  4856.7  144.91  4938.6  140.25  4968.9  140.38  4979.1  136.94
  4989.2  131.16  4996.3  130.39    4999  129.89  5002.3  130.39  5009.4  130.79
  5018.4  136.76  5023.5  134.67  5029.6   138.5  5039.7  140.27    5060  140.28
  5100.4  142.03  5231.9  150.88    5323  154.34  5393.8   155.9  5425.5  158.68
  5461.2  157.68  5515.5  160.16  5566.9  160.87  5661.4  160.44  5759.1  162.89
#Mann= 9 ,-1 , 0
  4417.7     .05       0  4519.2      .1       0  4591.1     .05       0
  4707.2      .1       0  4838.7     .05       0  4856.7      .1       0
  4996.3     .07       0  5002.3      .1       0  5515.5     .05       0
Bank Sta=4968.9,5039.7
XS Rating Curve= 0 ,0
Exp/Cntr=0.3,0.1

Type RM Length L Ch R = 1 ,28519   ,518,518,518
BEGIN DESCRIPTION:
UNT001 IN PECR 53.0
END DESCRIPTION:
XS GIS Cut Line= 3
      2290837.73     13251396.87      2290537.72     13250796.85
      2290537.72     13249996.89
#Sta/Elev= 30
  4337.1  170.87  4552.3  160.17  4605.4  155.28  4708.9  148.41  4851.4  150.79
  4891.6  153.52  4918.5  149.17  4926.9  144.56  4932.5  144.72  4949.2  140.37
  4971.6   137.6  4977.2  138.35  4985.6  131.36  4996.6  128.81  4999.3  128.31
  5002.6  128.81  5017.9  131.28  5026.3  136.37  5027.9  137.34  5047.9  138.81
  5222.2  144.36  5304.5  144.54  5494.5  147.22  5557.9  150.04  5677.9     161
  5707.9  161.02  5737.9  165.92  5767.9   166.9  5777.9  168.77  5807.9  170.62
#Mann= 8 ,-1 , 0
  4337.1     .05       0  4891.6      .1       0  4996.6     .07       0
  5002.6      .1       0  5026.3     .12       0  5222.2      .1       0
  5304.5     .12       0  5494.5      .1       0
Bank Sta=4977.2,5027.9
XS Rating Curve= 0 ,0
Exp/Cntr=0.3,0.1

Type RM Length L Ch R = 1 ,28001   ,540,540,540
BEGIN DESCRIPTION:
UNT001 IN PECR 52.0
END DESCRIPTION:
XS GIS Cut Line= 3
      2290887.72     13251346.82      2290987.72     13250546.85
      2291137.71      13249796.9
#Sta/Elev= 30
  4199.8  169.09  4323.2  161.79  4522.3  146.55  4658.7  145.06  4726.3     145
  4784.3  148.45  4844.7  148.82  4864.9  147.23  4915.3  139.13  4975.8  137.17
  4985.8   131.3  5000.5  127.98  5003.2  127.48  5006.5  127.98  5016.2  131.19
  5026.4  136.61  5069.5  137.89  5110.3  139.64  5169.2  142.51  5240.6  149.09
  5281.3  151.38  5301.7  154.39  5373.1  160.52  5444.5  164.55  5454.7  166.42
  5617.9   179.4  5679.1  186.09  5709.7  191.25  5740.3  194.01  5770.8  199.35
#Mann= 6 ,-1 , 0
  4199.8     .05       0  4658.7      .1       0  5000.5     .07       0
  5006.5      .1       0  5069.5     .12       0  5110.3      .1       0
Bank Sta=4975.8,5026.4
XS Rating Curve= 0 ,0
Exp/Cntr=0.3,0.1

Type RM Length L Ch R = 1 ,27461   ,499,499,499
BEGIN DESCRIPTION:
UNT001 IN PECR 51.0
END DESCRIPTION:
XS GIS Cut Line= 3
      2290963.51     13251481.19      2291580.67     13250555.45
      2291529.24      13250092.6
#Sta/Elev= 30
  4094.7  171.74  4267.9  163.19  4532.6  147.58  4598.4  145.59  4640.7  142.11
  4742.6  139.31    4802  141.32  4871.8  137.35  4943.9  137.42  4958.9  135.73
    4989     127  4998.3  125.84    5001  125.34  5004.3  125.84    5010  130.52
    5031  135.65  5061.1  136.62  5082.1  140.89  5097.1  142.38  5118.2  147.43
  5190.3  154.73  5246.1  157.55  5256.2  159.59  5326.6  162.48  5397.1  167.48
  5437.3  167.91  5467.5  170.19  5527.9  169.69    5558  173.31    5673  176.76
#Mann= 4 ,-1 , 0
  4094.7     .05       0    4802      .1       0  4998.3     .07       0
  5004.3      .1       0
Bank Sta=4943.9,5031
XS Rating Curve= 0 ,0
Exp/Cntr=0.3,0.1

Type RM Length L Ch R = 1 ,26962   ,573,573,573
BEGIN DESCRIPTION:
UNT001 IN PECR 50.0
END DESCRIPTION:
XS GIS Cut Line= 3
      2291087.69     13251846.89      2291837.72     13251046.85
      2292187.68     13250846.88
#Sta/Elev= 30
  3924.7  182.88  3990.7  177.84    3998  177.38  4122.5  168.92  4146.2  167.14
    4314  155.93  4504.8  145.69  4745.6  143.34  4853.2   138.5  4950.7  133.94
  4971.8  135.25  4979.1  132.48  4985.9  126.73  4997.1  124.19  4999.8  123.69
  5003.1  124.19  5014.2  128.23  5017.9  132.42  5024.2  132.42  5029.2  134.82
    5035  132.75  5050.8  134.12  5066.7  133.56  5131.5  138.23  5174.7  143.15
  5233.7  146.03  5276.9  150.97  5292.7  151.17  5298.5  153.02  5424.4  159.88
#Mann= 9 ,-1 , 0
  3924.7      .1       0  3990.7     .08       0    3998      .1       0
  4122.5     .05       0  4146.2      .1       0    4314     .05       0
  4853.2      .1       0  4997.1     .07       0  5003.1      .1       0
Bank Sta=4971.8,5017.9
XS Rating Curve= 0 ,0
Exp/Cntr=0.3,0.1

Type RM Length L Ch R = 1 ,26389   ,426,426,426
BEGIN DESCRIPTION:
UNT001 IN PECR 49.0
END DESCRIPTION:
XS GIS Cut Line= 2
      2291490.66     13252098.31       2292641.4     13251108.29
#Sta/Elev= 30
  4049.7  173.75  4074.8  171.89  4190.9  164.23  4211.8  161.64  4296.5  157.06
  4396.2  153.61  4474.1  152.48  4488.3  151.47  4576.3  149.58  4644.1   146.7
  4764.8  139.12  4863.7   136.7  4934.9  132.42  4953.4  132.87    4970  132.86
  4984.3  125.87  4995.6  123.88  4998.3  123.38  5001.6  123.88  5006.2  124.91
  5020.5  131.98  5090.7  135.19  5168.6  140.75  5279.2  143.38  5338.7  144.83
    5353  146.53  5367.2  145.69  5412.7  147.63  5445.1  148.87  5567.7  156.26
#Mann= 8 ,-1 , 0
  4049.7     .08       0  4074.8      .1       0  4576.3     .05       0
  4953.4      .1       0  4995.6     .07       0  5001.6      .1       0
  5279.2     .12       0  5412.7      .1       0
Bank Sta=4970,5020.5
XS Rating Curve= 0 ,0
Exp/Cntr=0.3,0.1

Type RM Length L Ch R = 1 ,25963   ,476,476,476
BEGIN DESCRIPTION:
UNT001 IN PECR 48.0
END DESCRIPTION:
XS GIS Cut Line= 3
      2292087.71     13252446.88      2292487.72     13251796.85
      2292687.74     13251446.82
#Sta/Elev= 30
  4236.4  181.51  4261.5  180.45  4267.6  180.06  4280.8  178.34  4295.1  173.13
    4308  170.86  4317.5  167.87  4381.5  159.36  4518.6  148.29  4619.5  143.53
    4655  142.82  4781.3  141.35  4837.1  137.07  4844.9  136.48    4934  131.99
  4964.4  133.04  4970.7  131.61  4993.7  121.72  4996.5  121.22  4999.7  121.72
  5007.6  123.61  5013.3  129.17  5018.6  130.22    5029  132.21  5050.8  131.43
  5072.3  132.61  5165.6  141.38  5305.6   152.5  5335.8  155.35  5402.8  158.94
#Mann= 14 ,-1 , 0
  4236.4      .1       0  4261.5     .05       0  4267.6     .08       0
  4381.5      .1       0  4619.5     .05       0    4655      .1       0
  4837.1     .05       0  4844.9      .1       0  4993.7     .07       0
  4999.7      .1       0  5018.6     .12       0    5029      .1       0
  5165.6     .12       0  5305.6      .1       0
Bank Sta=4970.7,5029
XS Rating Curve= 0 ,0
Exp/Cntr=0.3,0.1

Type RM Length L Ch R = 1 ,25487   ,402,402,402
BEGIN DESCRIPTION:
UNT001 IN PECR 47.0
END DESCRIPTION:
XS GIS Cut Line= 4
      2292679.93     13252484.04      2292859.95     13252291.16
      2292924.24     13251616.16      2292898.53     13251371.91
#Sta/Elev= 30
  4498.3  162.86  4560.4  159.99  4727.3  153.67  4776.5  152.79  4791.5  151.54
  4836.8   146.9  4846.8  144.85  4899.4  138.23  4917.1  134.94  4947.3  132.37
  4957.3   130.7  4977.4  130.33  4987.5  126.93  4997.4  120.93  4999.4  120.55
  5002.1  120.05  5005.4  120.55  5017.6  125.27  5030.5  128.98  5037.7  130.29
  5047.7  131.23  5067.8  130.12  5110.4  131.54  5128.1  133.17  5248.6  139.66
  5315.6  141.67  5528.6  150.72  5555.9  153.13  5600.4  155.43  5685.8  157.63
#Mann= 9 ,-1 , 0
  4498.3      .1       0  4560.4     .05       0  4727.3      .1       0
  4999.4     .07       0  5005.4      .1       0  5030.5     .12       0
  5315.6      .1       0  5528.6     .12       0  5555.9      .1       0
Bank Sta=4977.4,5037.7
XS Rating Curve= 0 ,0
Exp/Cntr=0.3,0.1

Type RM Length L Ch R = 1 ,25085   ,697,697,697
BEGIN DESCRIPTION:
UNT001 IN PECR 46.0
END DESCRIPTION:
XS GIS Cut Line= 3
      2293085.64     13252359.68      2293167.42     13252277.89
      2293817.23     13251278.18
#Sta/Elev= 30
  4680.9  148.36  4714.3  147.99  4766.6  147.34  4826.1  144.33  4940.9  129.63
  4964.8  128.72  4971.1  129.82    4977  128.35  4986.2   122.6  4997.6  120.48
  5000.3  119.98  5003.6  120.48  5035.5  128.92  5043.6  129.08  5049.5  126.02
  5062.8  128.39  5085.8  130.94  5100.9  131.05  5153.5  134.22  5203.3   135.4
  5251.8  134.88  5396.6  136.24  5477.6  136.41  5517.6  137.59  5671.6  144.03
  5728.9  148.12  5780.3  150.16  5837.6  155.22  5873.9  156.64  5988.9  164.63
#Mann= 10 ,-1 , 0
  4680.9      .1       0  4714.3     .05       0  4766.6      .1       0
  4997.6     .07       0  5003.6      .1       0  5035.5     .12       0
  5062.8      .1       0  5153.5     .12       0  5396.6      .1       0
  5517.6     .16       0
Bank Sta=4977,5035.5
XS Rating Curve= 0 ,0
Exp/Cntr=0.3,0.1

Type RM Length L Ch R = 1 ,24388   ,320,320,320
BEGIN DESCRIPTION:
UNT001 IN PECR 45.0
END DESCRIPTION:
XS GIS Cut Line= 3
      2293137.68     13252396.85      2293837.72     13252396.85
      2294237.67     13252296.87
#Sta/Elev= 30
  4309.4  145.98  4351.1  145.12  4454.8  144.83  4509.4  144.52  4649.4  139.31
  4789.4  136.54  4863.5  130.06  4899.4  127.61  4959.4   129.4  4969.4   128.8
  4979.4  126.55  4989.4  119.82  4996.4  118.63  4999.2  118.13  5002.4  118.63
  5006.9  120.27    5012  120.27  5027.5  127.66  5122.8  140.17  5192.4  147.56
  5197.6  147.22  5205.3  149.34  5233.6  153.63  5238.8  153.24  5246.5  155.66
  5267.1  157.99    5280  158.03  5316.1   163.2  5370.2  163.88  5421.7  162.07
#Mann= 6 ,-1 , 0
  4309.4     .05       0  4351.1      .1       0  4454.8     .05       0
  4863.5      .1       0  4996.4     .07       0  5002.4      .1       0
Bank Sta=4969.4,5027.5
XS Rating Curve= 0 ,0
Exp/Cntr=0.3,0.1

Type RM Length L Ch R = 1 ,24068   ,576,576,576
BEGIN DESCRIPTION:
UNT001 IN PECR 44.0
END DESCRIPTION:
XS GIS Cut Line= 3
      2292753.96     13253236.65      2294048.95      13252609.6
      2294193.55     13252437.89
#Sta/Elev= 30
  3801.7  171.18  3813.9  169.84  3816.5  169.74    3917  158.79  4034.5  149.54
  4185.4  139.47  4346.2  135.24    4473  131.94  4805.8  133.58  4912.7  126.95
  4963.5  126.51  4972.5  124.43  4980.5  119.75  4991.7  118.34  4994.5  117.84
  4997.7  118.34  5008.6  118.73  5025.7  127.83  5061.4  128.46    5099   136.7
  5121.6  138.84    5128  143.08  5138.6  144.26  5144.1  142.73  5150.3  145.63
  5166.7  146.45  5189.3  152.63  5205.8  154.59  5361.8  161.67    5465  161.68
#Mann= 9 ,-1 , 0
  3801.7     .08       0  3813.9     .05       0  3816.5      .1       0
  4034.5     .05       0  4185.4      .1       0  4346.2     .05       0
    4473      .1       0  4991.7     .07       0  4997.7      .1       0
Bank Sta=4963.5,5025.7
XS Rating Curve= 0 ,0
Exp/Cntr=0.3,0.1

Type RM Length L Ch R = 1 ,23492   ,585,585,585
BEGIN DESCRIPTION:
UNT001 IN PECR 43.0
END DESCRIPTION:
XS GIS Cut Line= 3
      2293617.26     13253772.89       2294167.1     13252882.24
      2294212.45     13252501.22
#Sta/Elev= 30
  4409.4  167.04  4573.6  161.27  4662.3  153.57  4704.9  148.52  4720.3  145.52
  4741.5  144.06  4747.4  142.54  4820.7  134.61    4900   127.8  4973.3  124.62
  4980.6  122.33  4991.6  116.64  4994.3  116.14  4997.6  116.64  5004.1  117.06
  5025.3  121.88  5031.2  125.25  5040.8  125.72  5089.2  126.72  5141.2  131.74
  5162.5  132.09  5192.1  134.51  5312.7  134.86  5456.1  136.71  5562.2     143
  5587.8  145.83  5602.5  145.92  5670.4   152.8    5753  157.18  5839.8  160.09
#Mann= 5 ,-1 , 0
  4409.4      .1       0  4991.6     .07       0  4997.6      .1       0
  5040.8     .12       0  5312.7      .1       0
Bank Sta=4973.3,5031.2
XS Rating Curve= 0 ,0
Exp/Cntr=0.3,0.1

Type RM Length L Ch R = 1 ,22907   ,643,643,643
BEGIN DESCRIPTION:
UNT001 IN PECR 42.0
END DESCRIPTION:
XS GIS Cut Line= 4
      2293992.57     13254089.11      2294226.91     13253915.53
      2294643.58     13253142.96      2294739.06     13252752.35
#Sta/Elev= 30
  4331.6  159.75  4374.9  158.72  4428.4  158.04  4550.6  153.49  4600.1   150.3
  4757.1  139.66  4822.8   134.1  4837.6  133.95  4926.6  125.02  4955.5  123.78
  4962.6  123.66  4976.1  121.45    4995  116.12  4997.7  115.62    5001  116.12
    5008  117.56  5014.2  122.36  5019.9   123.8  5030.4  125.16  5096.1  124.17
  5123.7  125.31  5139.9  127.12  5227.4  129.29  5299.2  132.42    5435  138.02
  5548.5     144  5610.2  145.13  5630.8  147.45  5832.9  157.26  5903.1  159.74
#Mann= 8 ,-1 , 0
  4331.6     .05       0  4374.9      .1       0  4428.4     .05       0
  4600.1      .1       0  4955.5     .12       0    4995     .07       0
    5001     .12       0  5299.2      .1       0
Bank Sta=4962.6,5019.9
XS Rating Curve= 0 ,0
Exp/Cntr=0.3,0.1

Type RM Length L Ch R = 1 ,22264   ,434,434,434
BEGIN DESCRIPTION:
UNT001 IN PECR 41.0
END DESCRIPTION:
XS GIS Cut Line= 3
      2294921.35     13254618.66      2295008.16     13254080.46
       2295034.2     13252925.91
#Sta/Elev= 30
    4042  164.93  4165.4  159.93  4374.2  147.57  4509.8  140.84  4540.2  140.25
  4586.5   137.1  4715.1  132.77  4800.8  128.46  4834.7  123.79  4870.8   121.9
  4898.1  122.35  4920.8  122.86  4940.9   121.5  4970.9  122.94  4990.9     118
  4997.9  115.11  5000.6  114.61  5003.9  115.11  5010.9  115.64  5020.9  121.67
  5030.9  124.83  5070.9  124.25  5100.9  127.69  5110.9  126.94  5147.4  128.18
  5190.9  128.79  5310.9  136.18    5471  143.54    5651  153.67    5742  156.35
#Mann= 8 ,-1 , 0
    4042     .05       0  4374.2      .1       0  4715.1     .05       0
  4834.7     .16       0  4898.1     .05       0  4997.9     .04       0
  5003.9     .05       0  5147.4      .1       0
Bank Sta=4970.9,5030.9
XS Rating Curve= 0 ,0
Exp/Cntr=0.3,0.1

Type RM Length L Ch R = 1 ,21830   ,646,646,646
BEGIN DESCRIPTION:
UNT001 IN PECR 40.0
END DESCRIPTION:
XS GIS Cut Line= 3
       2295173.1     13254601.27      2295329.34     13254002.33
      2295676.13     13252970.64
#Sta/Elev= 30
  4138.4  157.71  4177.8   156.3  4253.6  156.13    4329  152.41    4422  144.74
  4491.3  141.35  4496.5  140.07  4587.3  137.19  4653.2   133.7  4713.6  133.47
  4794.5  133.05  4831.2  131.69  4865.3  128.55    4932  120.97  4968.5  122.17
  4974.2  122.01  4983.6  119.28  4988.8  119.48  4995.3  113.82  5002.8  113.01
  5005.6  112.51  5008.8  113.01  5015.1  120.24  5020.4  119.43  5026.9  121.63
  5117.7  121.41  5195.7   125.3    5304  124.92  5644.1  132.61  5845.8  144.13
#Mann= 8 ,-1 , 0
  4138.4      .1       0  4713.6     .12       0  4865.3     .05       0
  4968.5     .16       0  5002.8     .07       0  5008.8     .16       0
  5117.7      .1       0  5644.1     .05       0
Bank Sta=4974.2,5026.9
XS Rating Curve= 0 ,0
Exp/Cntr=0.3,0.1

Type RM Length L Ch R = 1 ,21184   ,594,594,594
BEGIN DESCRIPTION:
UNT001 IN PECR 39.0
END DESCRIPTION:
XS GIS Cut Line= 2
      2296093.23     13254340.89       2295971.7     13252986.73
#Sta/Elev= 30
  4320.4  163.46  4438.9  160.89  4550.1  154.59  4605.6  149.95  4645.7  145.74
  4675.9  141.12  4726.1  136.92  4746.1  133.97  4841.8  124.38  4883.6  119.93
  4941.3  119.45    4967  121.32  4977.1  120.32  4987.1  117.63  4996.8  111.74
  4999.5  111.24  5002.8  111.74  5007.2  112.19  5017.2  117.49  5027.3   120.1
  5047.3  119.56  5073.8  121.28  5137.7  126.24  5177.9  127.76  5288.3  127.37
  5364.8  128.97  5459.9   134.5  5519.2  138.87  5569.4  140.65    5680  147.31
#Mann= 8 ,-1 , 0
  4320.4      .1       0  4841.8     .05       0  4941.3     .16       0
  4996.8     .07       0  5002.8     .16       0  5073.8      .1       0
  5364.8     .16       0  5459.9      .1       0
Bank Sta=4977.1,5027.3
XS Rating Curve= 0 ,0
Exp/Cntr=0.3,0.1

Type RM Length L Ch R = 1 ,20590   ,476,476,476
BEGIN DESCRIPTION:
UNT001 IN PECR 38.0
END DESCRIPTION:
XS GIS Cut Line= 3
      2296537.72     13254096.88      2296587.72     13253696.85
      2296637.72     13253146.86
#Sta/Elev= 30
  4586.2  152.37  4616.5  148.96  4748.8  140.58  4785.3  136.88  4790.3  137.67
    4848  132.64  4900.2  128.38  4928.9  125.51  4947.2  122.48  4959.1  122.19
  4969.2  120.49  4979.3  118.12  4986.8  114.01  4991.8  114.01  4996.4  110.94
  4999.1  110.44  5002.4  110.94  5009.4  111.42  5029.5   117.6  5039.5  118.63
  5059.6  120.04  5119.9  117.93  5170.1   117.9  5190.2   120.7  5260.5  123.52
  5290.6  126.31    5391  131.38  5460.8  138.12  5464.6  138.33  5541.6     144
#Mann= 9 ,-1 , 0
  4586.2      .1       0  4748.8     .08       0    4848      .1       0
  4900.2     .08       0  4947.2      .1       0  4996.4     .07       0
  5002.4      .1       0  5460.8     .16       0  5464.6      .1       0
Bank Sta=4969.2,5039.5
XS Rating Curve= 0 ,0
Exp/Cntr=0.3,0.1

Type RM Length L Ch R = 1 ,20114   ,671,671,671
BEGIN DESCRIPTION:
UNT001 IN PECR 37.0
END DESCRIPTION:
XS GIS Cut Line= 3
      2296692.19     13254175.94      2296969.96     13253941.57
      2297204.34     13253004.06
#Sta/Elev= 30
  4301.9  152.25    4412  147.57  4560.3  143.41  4681.2  136.68  4760.1  130.29
  4861.2  124.35  4882.2  121.42  4923.4  118.08  4969.8  118.01  4979.4   116.9
  4986.7  109.32  4989.5  108.82  4992.7  109.32    5000  109.37  5005.9  114.52
    5011  114.09  5014.7  115.55  5020.7  117.92  5080.3  116.33  5088.3   115.1
  5113.4  115.31  5170.8   123.2  5278.4  132.27  5335.7  138.91  5371.1  140.89
    5377   142.2  5494.8  148.18  5505.8  149.81  5577.3  154.43  5631.7  156.73
#Mann= 7 ,-1 , 0
  4301.9      .1       0  4760.1     .08       0  4861.2      .1       0
  4986.7     .07       0  4992.7      .1       0  5014.7     .16       0
  5080.3      .1       0
Bank Sta=4969.8,5014.7
XS Rating Curve= 0 ,0
Exp/Cntr=0.3,0.1

Type RM Length L Ch R = 1 ,19443   ,510,510,510
BEGIN DESCRIPTION:
UNT001 IN PECR 36.0
END DESCRIPTION:
XS GIS Cut Line= 3
      2297721.29     13254312.59      2297587.32     13253332.93
       2297412.1     13252899.05
#Sta/Elev= 30
  4469.8  148.66  4526.1  146.82  4537.1  145.54  4596.7  143.02  4694.5   135.4
  4768.3  130.62    4826  125.49  4838.9  125.71  4869.2  122.26  4903.3  121.27
  4930.2  119.18  4970.1   116.3  4980.6  116.36  4990.3  109.22  4997.4   108.3
  5000.2   107.8  5003.4   108.3  5030.7  116.71  5115.4  116.18  5141.7  115.36
    5172  116.18  5192.2   117.9  5197.3  119.63  5262.8  123.74  5323.4  124.23
  5404.1   127.2  5691.6  146.38  5810.2  151.97  5816.8  153.14  5926.5  158.95
#Mann= 6 ,-1 , 0
  4469.8     .05       0  4694.5      .1       0  4930.2     .16       0
  4997.4     .07       0  5003.4     .16       0  5115.4      .1       0
Bank Sta=4980.6,5030.7
XS Rating Curve= 0 ,0
Exp/Cntr=0.3,0.1

Type RM Length L Ch R = 1 ,18933   ,522,522,522
BEGIN DESCRIPTION:
UNT001 IN PECR 35.0
END DESCRIPTION:
XS GIS Cut Line= 2
      2298219.49     13254038.77      2297902.72     13252781.77
#Sta/Elev= 30
  4619.4  143.36  4683.1  142.26  4782.7   133.8  4837.9  127.75  4847.4  125.51
  4888.5  120.66  4893.7  118.87  4899.8  118.23  4934.7  116.75  4941.1  114.98
  4961.7  114.13  4975.8   114.9  4982.3  108.71  4993.7  106.64  4999.9   106.3
  5002.7   105.8  5005.9   106.3  5011.8  108.22  5023.6  115.08  5052.8  115.81
  5116.4  113.83  5235.2  118.95  5332.9   119.4  5405.1  122.65  5496.5   122.6
  5580.5   123.9  5627.8   126.1  5650.9  127.35  5792.4  137.23  5915.7  144.62
#Mann= 9 ,-1 , 0
  4619.4      .1       0  4782.7     .16       0  4993.7      .1       0
  4999.9     .07       0  5005.9      .1       0  5235.2     .16       0
  5496.5      .1       0  5627.8     .16       0  5650.9      .1       0
Bank Sta=4975.8,5023.6
XS Rating Curve= 0 ,0
Exp/Cntr=0.3,0.1

Type RM Length L Ch R = 1 ,18411   ,463,463,463
BEGIN DESCRIPTION:
UNT001 IN PECR 34.0
END DESCRIPTION:
XS GIS Cut Line= 4
      2298446.05       13253918.      2298526.61      13253590.7
      2298587.03     13252976.46      2298707.35     13252680.67
#Sta/Elev= 30
  4447.6  142.03    4475  143.55  4514.4  143.31    4515  143.29  4784.1  125.64
    4879  123.48    4889  121.98  4899.1  118.24  4909.1  117.69  4919.2  115.06
    4933  113.46  4969.4  114.03  4989.5  108.52  4996.5   104.3  4999.3   103.8
  5002.5   104.3  5009.6  106.75  5019.6  112.49  5029.7  114.03    5044  113.65
  5079.9   112.3  5240.7  116.98  5465.4  138.73  5524.4  141.38    5602  142.73
  5607.4  143.95  5655.5  144.24  5660.9  145.61  5679.6   145.2  5721.2  147.57
#Mann= 7 ,-1 , 0
  4447.6      .1       0  4514.4     .16       0    4515      .1       0
    4933     .16       0  4996.5     .07       0  5002.5     .16       0
    5044      .1       0
Bank Sta=4969.4,5029.7
XS Rating Curve= 0 ,0
Exp/Cntr=0.3,0.1

Type RM Length L Ch R = 1 ,17948   ,627,627,627
BEGIN DESCRIPTION:
UNT001 IN PECR 33.0
END DESCRIPTION:
XS GIS Cut Line= 4
      2299014.98     13253963.22      2298989.81     13253117.43
      2298874.01     13252820.38      2298773.33     13252634.13
#Sta/Elev= 30
  4304.2  134.69  4480.6  128.41  4620.7  117.85  4672.3  115.79  4728.2  114.62
  4770.8   116.8  4800.8  116.83  4890.8  111.45    4928  112.67  4950.8  112.38
  4970.9  110.06  4980.9  106.19  4997.9  104.45  5000.6  103.95  5003.9  104.45
  5020.9  111.75  5054.1  111.91  5067.2  113.83  5130.9  121.37  5148.1  125.72
  5161.7  126.69  5168.5  128.78  5183.2  129.34    5193  131.47  5198.3   130.7
  5222.8  134.05  5228.2  133.29  5336.9  134.76  5529.7  143.57  5680.9  148.84
#Mann= 7 ,-1 , 0
  4304.2      .1       0  4672.3     .16       0  4728.2      .1       0
    4928     .16       0  4997.9     .07       0  5003.9     .16       0
  5067.2      .1       0
Bank Sta=4950.8,5020.9
XS Rating Curve= 0 ,0
Exp/Cntr=0.3,0.1

Type RM Length L Ch R = 1 ,17321   ,646,646,646
BEGIN DESCRIPTION:
UNT001 IN PECR 32.0
END DESCRIPTION:
XS GIS Cut Line= 3
      2299664.46     13254008.56      2299528.52     13252860.66
      2299468.09     13252674.34
#Sta/Elev= 30
  4403.6  140.15    4585  130.58  4687.3  121.52  4783.5  115.59  4902.7  109.83
  4949.1  108.99  4959.2  110.95  4969.2  111.55  4973.8  110.17  4996.4  102.76
  4999.2  102.26  5002.4  102.76    5009   104.4  5014.1  104.43  5019.6  110.76
    5080  110.11  5110.2  113.34  5136.2  114.33  5184.7  114.43  5210.9  115.75
  5251.2  115.42  5301.5  117.09  5355.3  119.51    5362  120.66  5432.4  124.84
  5438.1  126.48  5443.2  125.62  5558.9  134.13  5674.7  139.47  5755.4  141.16
#Mann= 7 ,-1 , 0
  4403.6      .1       0  4783.5     .16       0  4902.7      .1       0
  4973.8     .16       0  4996.4     .07       0  5002.4     .16       0
  5136.2      .1       0
Bank Sta=4969.2,5019.6
XS Rating Curve= 0 ,0
Exp/Cntr=0.3,0.1

Type RM Length L Ch R = 1 ,16675   ,311,311,311
BEGIN DESCRIPTION:
UNT001 IN PECR 31.0
END DESCRIPTION:
XS GIS Cut Line= 3
      2300559.76     13253609.27      2300350.41     13253366.42
      2299647.08     13252562.61
#Sta/Elev= 30
  4390.6  162.15  4441.6  159.11  4470.4  157.34  4570.2  149.81  4663.1  143.84
  4670.8  144.48  4748.6  136.83  4762.8  133.63  4818.8  126.68  4861.5  118.01
  4875.8  116.86    4890  113.96    4910   112.9  4925.1  110.15  4953.6   108.3
  4975.4  108.97  4975.9  108.85    5000  102.33  5002.7  101.83    5006  102.33
  5024.8  109.56    5039  109.87  5045.1  108.83  5067.5   107.3  5088.4  107.43
  5285.7  114.73  5414.9   121.9  5506.9  129.12    5599  134.67  5779.3  139.55
#Mann= 10 ,-1 , 0
  4390.6     .05       0  4441.6      .1       0  4470.4     .05       0
  4570.2      .1       0    4910     .16       0  4975.9      .1       0
    5000     .07       0    5006      .1       0  5045.1     .16       0
  5285.7      .1       0
Bank Sta=4975.4,5024.8
XS Rating Curve= 0 ,0
Exp/Cntr=0.3,0.1

Type RM Length L Ch R = 1 ,16364   ,633,633,633
BEGIN DESCRIPTION:
UNT001 IN PECR 30.0
END DESCRIPTION:
XS GIS Cut Line= 3
      2300737.75     13253246.88      2300387.72     13252946.85
      2299837.69     13252346.82
#Sta/Elev= 30
  4510.9  154.47  4553.2  152.54  4575.1  149.53  4616.9  146.83  4638.8  143.55
  4645.4  140.46  4653.1  139.33  4695.3  136.91  4773.8  128.04  4780.4  128.84
  4787.5  125.78  4893.4  111.78  4901.1  109.47  4946.8   107.7    4979   108.5
  4993.2  101.31  5004.4  100.49  5007.1   99.99  5010.4  100.49  5021.6  107.52
  5052.1  108.51  5087.7  107.15  5318.8  115.31  5481.3  123.54  5495.7  125.71
  5524.1  125.52  5665.3   133.8  5701.1  137.79  5776.4  138.04  5785.9  139.41
#Mann= 8 ,-1 , 0
  4510.9      .1       0  4946.8     .16       0  5004.4     .07       0
  5010.4     .16       0  5052.1      .1       0  5087.7     .16       0
  5481.3      .1       0  5776.4     .08       0
Bank Sta=4979,5021.6
XS Rating Curve= 0 ,0
Exp/Cntr=0.3,0.1

Type RM Length L Ch R = 1 ,15731   ,598,598,598
BEGIN DESCRIPTION:
UNT001 IN PECR 29.0
END DESCRIPTION:
XS GIS Cut Line= 4
      2301187.04     13253190.63      2300989.12     13252607.29
      2300301.62     13252086.46      2299775.58     13252060.41
#Sta/Elev= 30
  4125.4  157.43  4192.7  155.11    4231  151.44  4293.8  148.27  4445.5  134.97
  4678.5  124.83  4749.9  120.72  4770.7  118.25  4785.3  118.47  4849.8  113.03
  4885.2  108.59  4938.7  105.47  4949.5  105.64  4978.8   106.2  5003.6   99.89
  5006.4   99.39  5009.6   99.89  5028.7  106.61  5070.3  105.38  5119.7  106.18
  5174.4  108.15  5213.9  110.46    5290  112.07  5463.5  114.87  5578.1  121.76
  5657.9   127.6  5788.1  132.42  5991.7  140.24  6009.5   140.9  6130.6  144.75
#Mann= 12 ,-1 , 0
  4125.4      .1       0  4938.7     .16       0  4949.5     .05       0
  5003.6     .04       0  5009.6     .05       0  5119.7      .1       0
  5174.4     .05       0    5290      .1       0  5578.1     .05       0
  5788.1      .1       0  5991.7     .05       0  6009.5      .1       0
Bank Sta=4978.8,5028.7
XS Rating Curve= 0 ,0
Exp/Cntr=0.3,0.1

Type RM Length L Ch R = 1 ,15133   ,472,472,472
BEGIN DESCRIPTION:
UNT001 IN PECR 28.0
END DESCRIPTION:
XS GIS Cut Line= 4
      2301690.08     13252051.86      2301330.05     13252143.96
      2300559.74     13251566.22      2300350.39     13251214.52
#Sta/Elev= 30
  4326.6  132.98  4341.2  132.65  4421.9  130.85  4442.5   132.1  4473.5  128.41
  4576.7   127.7  4726.1  121.47  4836.1   111.6  4904.6  106.64  4910.6  105.41
  4919.1   104.3  4933.7   99.89  4945.3   99.02  4948.1   98.52  4951.3   99.02
    4990   99.13  5026.1  104.11  5048.3  105.95  5083.7  106.62  5119.1  104.63
  5150.7  104.25  5204.6  106.27  5462.9  108.88  5562.9  114.24  5619.1  118.82
  5644.5  119.57  5830.2   132.7  5968.4  139.44  5989.8  141.53  6070.4  143.81
#Mann= 9 ,-1 , 0
  4326.6      .1       0  4341.2     .05       0  4576.7      .1       0
  4836.1     .05       0  4910.6      .1       0  4945.3     .07       0
  4951.3      .1       0  5150.7     .05       0  5644.5      .1       0
Bank Sta=4904.6,5048.3
XS Rating Curve= 0 ,0
Exp/Cntr=0.3,0.1

Type RM Length L Ch R = 1 ,14661   ,397,397,397
BEGIN DESCRIPTION:
UNT001 IN PECR 27.0
END DESCRIPTION:
XS GIS Cut Line= 4
      2301757.08     13251934.63      2301505.89     13251767.17
      2300986.76     13251206.18      2300836.03     13250913.09
#Sta/Elev= 30
  4401.8  134.74  4435.7  133.58  4521.2  129.86  4536.1  130.73  4545.1  128.74
  4557.3   127.8  4622.1  125.45  4658.1   122.7  4680.3  119.65    4706   118.6
  4723.8  116.18  4781.5  113.52  4788.6  112.69  4858.2  108.14  4900.7  104.27
  4929.1  103.52  4951.7  104.41  4971.6  104.87  4989.6   99.19  4992.3   98.69
  4995.6   99.19  5014.1  104.24  5099.2  103.12  5192.5  104.93  5268.7  107.83
  5410.4  116.82  5639.1  129.15  5642.7  129.37  5725.9  133.01  5797.6  134.68
#Mann= 12 ,-1 , 0
  4401.8     .05       0  4435.7      .1       0  4622.1     .05       0
  4658.1      .1       0  4781.5     .05       0  4788.6      .1       0
  4951.7     .12       0  4989.6     .07       0  4995.6     .12       0
  5192.5      .1       0  5639.1     .05       0  5642.7      .1       0
Bank Sta=4971.6,5014.1
XS Rating Curve= 0 ,0
Exp/Cntr=0.3,0.1

Type RM Length L Ch R = 1 ,14264   ,432,432,432
BEGIN DESCRIPTION:
UNT001 IN PECR 26.0
END DESCRIPTION:
XS GIS Cut Line= 3
      2302033.38     13251691.81      2301824.06     13251432.25
      2300903.02     13250804.27
#Sta/Elev= 30
  4256.4  127.93  4370.5  123.62  4455.5  121.28  4512.8  117.67  4527.2   116.1
  4570.4   115.2  4647.9   111.1  4785.5  107.19    4841  104.24  4892.6  102.73
  4914.2  102.51  4929.1  103.86    4965  104.29  4979.9  102.91  4994.9   98.45
    5006   97.55  5008.8   97.05    5012   97.55  5015.8  104.01  5030.8   104.2
  5051.7  102.58  5087.6  102.01  5123.6  103.32  5144.6  104.86    5360  122.35
  5432.6  125.31  5478.5  126.38  5569.4  128.83  5662.6  132.61  5704.6  133.44
#Mann= 7 ,-1 , 0
  4256.4     .05       0    4841      .1       0  4892.6     .12       0
    5006     .07       0    5012     .12       0  5144.6     .05       0
  5478.5      .1       0
Bank Sta=4965,5015.8
XS Rating Curve= 0 ,0
Exp/Cntr=0.3,0.1

Type RM Length L Ch R = 1 ,13832   ,452,452,452
BEGIN DESCRIPTION:
UNT001 IN PECR 25.0
END DESCRIPTION:
XS GIS Cut Line= 3
      2302175.74     13251055.48      2302066.88     13250946.62
      2301045.34     13250653.55
#Sta/Elev= 30
  4496.3  122.55  4578.8   124.2    4600  123.72  4652.4  120.49  4753.4  111.06
  4860.4  103.35  4923.2  101.69  4962.2  103.06  4971.9  102.58  4982.3  101.62
  4987.7   98.62  4990.4   98.12  4993.7   98.62  5023.9  101.44  5029.6  102.91
  5044.7  103.52  5085.8  101.99    5136  101.49  5200.8  106.72  5252.9   112.9
  5286.6  113.09  5366.8  116.29  5419.2   117.3  5450.4  119.27  5504.6  119.95
  5544.1  121.36  5564.9  123.28  5596.1  123.57  5628.1  125.36    5713  130.49
#Mann= 7 ,-1 , 0
  4496.3     .05       0  4860.4     .12       0  4987.7     .07       0
  4993.7     .12       0  5085.8      .1       0  5366.8     .05       0
  5628.1      .1       0
Bank Sta=4971.9,5029.6
XS Rating Curve= 0 ,0
Exp/Cntr=0.3,0.1

Type RM Length L Ch R = 1 ,13380   ,614,614,614
BEGIN DESCRIPTION:
UNT001 IN PECR 24.0
END DESCRIPTION:
XS GIS Cut Line= 3
      2302242.74     13250687.09      2302158.98     13250594.95
       2301028.6     13249883.23
#Sta/Elev= 30
  4604.3  122.68  4650.4  122.84  4699.8  118.39  4765.8  117.45  4793.1  115.71
  4826.3  109.55  4902.6  101.95    4945  100.44  4975.6  102.04  4985.4  101.17
  4993.8   99.11  4996.5   98.61  4999.8   99.11  5002.7  100.87  5012.1  102.19
    5018  100.55  5025.7  103.48  5033.6  104.37  5039.2  104.43  5048.6  101.66
  5069.8  100.92  5155.7  100.99  5498.3  106.48  5510.2  105.58  5686.7  112.37
  5798.7  119.56  5817.4  119.92  5857.3  123.51  5990.5  131.95  6064.6  135.25
#Mann= 8 ,-1 , 0
  4604.3     .05       0  4826.3      .1       0  4985.4     .12       0
  4993.8     .07       0  4999.8     .12       0  5033.6      .1       0
  5798.7     .05       0  5857.3      .1       0
Bank Sta=4975.6,5012.1
XS Rating Curve= 0 ,0
Exp/Cntr=0.3,0.1

Type RM Length L Ch R = 1 ,12766   ,528,528,528
BEGIN DESCRIPTION:
UNT001 IN PECR 23.0
END DESCRIPTION:
XS GIS Cut Line= 3
      2302870.89     13250630.02       2302104.3     13249865.44
      2301115.84     13249642.01
#Sta/Elev= 30
  3917.3  117.84  3992.5  118.65  4310.7  108.27  4374.3  108.85  4381.4  110.96
  4395.5  111.01  4459.2  108.13  4480.4  111.05  4586.5   107.1  4855.2  106.25
  4932.9   99.91  4968.3  100.62  4992.5   96.81  4995.2   96.31  4998.5   96.81
  5008.4   98.34  5014.1   99.51  5067.2   99.67  5191.3  100.33  5240.2  102.64
  5291.2  102.81  5423.2  102.41    5539  108.26  5570.6  111.74  5613.1   114.1
  5642.4  115.13  5673.1  119.24  5713.1  121.23  5847.4  129.92  6013.4  138.41
#Mann= 9 ,-1 , 0
  3917.3     .05       0  4992.5     .03       0  4998.5     .05       0
  5008.4      .1       0  5067.2     .05       0  5291.2     .12       0
    5539      .1       0  5613.1     .08       0  5713.1      .1       0
Bank Sta=4968.3,5014.1
XS Rating Curve= 0 ,0
Exp/Cntr=0.3,0.1

Type RM Length L Ch R = 1 ,12238   ,592,592,592
BEGIN DESCRIPTION:
UNT001 IN PECR 22.0
END DESCRIPTION:
XS GIS Cut Line= 3
      2302837.73     13250496.89      2302337.72     13249396.85
      2301587.74     13248596.87
#Sta/Elev= 30
  3792.3  118.76  3898.9  116.36  4068.2   105.4  4117.7  103.35  4485.5   99.72
  4595.5   98.84  4675.5   98.92    4715  103.12  4773.3  105.38  4790.8  101.66
  4815.5  101.77  4911.7   98.52  4945.7  101.08  4978.7   99.84  5004.7   92.85
  5007.5   92.35  5010.7   92.85  5014.6   97.45    5036   97.53  5042.9  100.69
  5071.2   98.65  5095.9   99.92  5283.7  101.65  5323.3  106.33  5354.5  103.88
  5411.2  104.09  5446.4   108.8  5601.8  117.08  5608.7  117.29  6097.2  156.24
#Mann= 12 ,-1 , 0
  3792.3     .05       0  4068.2      .1       0  4117.7     .05       0
  4485.5     .12       0  4595.5      .1       0  4815.5     .05       0
  5004.7    .035       0  5010.7     .05       0  5095.9     .12       0
  5323.3      .1       0  5601.8     .05       0  5608.7      .1       0
#XS Ineff= 2 , 0
            4775  105.51
Permanent Ineff=
       F       F
Bank Sta=4978.7,5042.9
XS Rating Curve= 0 ,0
Exp/Cntr=0.3,0.1

Type RM Length L Ch R = 1 ,11646   ,393,393,393
BEGIN DESCRIPTION:
UNT001 IN PECR 21.0
END DESCRIPTION:
XS GIS Cut Line= 3
      2303078.91     13250645.52       2302716.1     13248824.38
      2302154.09     13248297.93
#Sta/Elev= 30
  3309.6  116.61  3420.4   115.6  3490.7   111.8  3495.8  113.36  3532.6  113.73
  3546.9  113.26    3553  109.06  3573.3  107.08  3683.2  106.17  3736.5  106.42
  3767.1  101.83  3879.2  100.04    3920  100.52  3950.5  103.41  4050.4  102.63
  4522.6  100.37  4701.2   98.31  4977.2   98.19  4994.2   95.27  4997.9   94.87
  5000.6   94.37  5003.9   94.87  5028.3   97.78  5106.5  101.67  5173.4  106.38
  5207.8  108.34    5360  119.17  5545.8  134.17  5807.6  148.31  5936.6  159.63
#Mann= 12 ,-1 , 0
  3309.6     .05       0  3683.2      .1       0  4050.4     .05       0
  4522.6      .1       0  4701.2     .12       0  4994.2      .1       0
  4997.9     .07       0  5003.9      .1       0  5106.5     .12       0
  5173.4      .1       0  5207.8     .05       0    5360      .1       0
#XS Ineff= 2 , 0
         4005.68  104.02
Permanent Ineff=
       F       F
Bank Sta=4977.2,5028.3
XS Rating Curve= 0 ,0
Exp/Cntr=0.3,0.1

Type RM Length L Ch R = 1 ,11253   ,702,702,702
BEGIN DESCRIPTION:
UNT001 IN PECR 20.0
END DESCRIPTION:
XS GIS Cut Line= 4
      2303249.63     13250638.35       2303342.1     13249635.33
      2302993.53     13248426.01       2302495.6     13248041.89
#Sta/Elev= 30
  3200.5   110.1  3292.4  109.99  3340.3  107.29  3458.8     106  3656.6   101.9
  3770.3  101.23  3824.6  102.17  4216.6   97.48    4356   97.74  4633.5   99.58
  4744.2    97.2  4817.2   96.26  4889.7   97.38  4934.7   95.82  4962.2   97.29
 4970.74   97.28  4998.1   95.02  5000.9   94.52  5004.1   95.02  5012.4   96.12
  5028.4    97.5  5090.8   96.24  5151.9    99.1  5309.3  102.75  5446.9  109.46
  5605.4  117.62  5640.5  118.89    5655  121.21  5962.1  144.04  6095.2  148.04
#Mann= 14 ,-1 , 0
  3200.5     .08       0  3458.8     .05       0  3656.6      .1       0
  3770.3     .05       0    4356     .12       0  4633.5      .1       0
  4744.2     .12       0  4962.2     .05       0  4998.1    .035       0
  5004.1     .05       0  5012.4     .12       0  5151.9      .1       0
  5446.9     .05       0  5605.4      .1       0
#XS Ineff= 2 , 0
         3833.24  102.24
Permanent Ineff=
       F       F
Bank Sta=4970.74,5028.4
XS Rating Curve= 0 ,0
Exp/Cntr=0.3,0.1

Type RM Length L Ch R = 1 ,10551   ,294,294,294
BEGIN DESCRIPTION:
UNT001 IN PECR 19.0
END DESCRIPTION:
XS GIS Cut Line= 5
      2303299.42     13250538.78      2303783.15     13248966.65
      2303811.61     13248063.21      2303619.54     13247686.19
      2303164.23     13247358.93
#Sta/Elev= 30
  3066.5   107.4  3229.1  107.06  3331.5  105.82    3489  103.19  3549.2   99.73
    3946   97.81  3986.2   97.83  4468.6    99.3  4669.3   98.44  4750.2   95.24
  4778.2    94.7  4780.9    94.2  4784.2    94.7  4971.3   95.87  5031.3   96.29
  5199.6   95.59  5330.5   97.61    5637  108.93  5653.7  111.64  5659.3   109.6
  5703.7  109.86  5912.2  117.39  6020.9  119.77  6146.8   121.8  6265.1  127.65
  6323.3  130.86  6499.9  142.45  6502.9  142.56  6570.2  147.01  6599.1  146.27
#Mann= 17 ,-1 , 0
  3066.5     .08       0  3229.1     .05       0  3331.5     .08       0
    3946      .1       0  3986.2     .08       0  4750.2     .05       0
  4778.2     .03       0  4784.2     .05       0  5199.6     .12       0
  5330.5      .1       0  5912.2     .08       0  6020.9      .1       0
  6146.8     .08       0  6265.1      .1       0  6323.3     .08       0
  6499.9      .1       0  6502.9     .08       0
#XS Ineff= 2 , 0
            4300   99.91
Permanent Ineff=
       F       F
Bank Sta=4971.3,5031.3
XS Rating Curve= 0 ,0
Exp/Cntr=0.3,0.1

Type RM Length L Ch R = 1 ,10257   ,592,592,592
BEGIN DESCRIPTION:
UNT001 IN PECR 18.0
END DESCRIPTION:
XS GIS Cut Line= 5
      2303342.11     13250695.27      2304010.79     13249087.58
      2304131.72      13248006.3      2303932.54     13247750.21
      2303285.95     13247281.26
#Sta/Elev= 30
  2749.6  110.37  2872.1  108.89  3083.5  104.51  3302.6  102.21  3506.2   99.59
  3577.6   98.51    3919   96.68  4140.3   96.22  4351.7   96.06  4457.3   97.28
  4657.6   97.86  4756.6   93.41  4855.7   94.96  4964.5   95.38  5001.7   91.98
  5004.5   91.48  5007.7   91.98  5034.9    95.2  5165.7   92.71  5305.6   96.85
    5614  107.32  5767.2     113    5788  114.86  5794.4  118.15  5931.1  124.49
  5976.1  123.72  6141.5  124.84  6283.6  125.49  6481.6  131.73    6702  143.91
#Mann= 20 ,-1 , 0
  2749.6     .05       0  2872.1      .1       0  3083.5     .05       0
  3302.6      .1       0  3506.2     .08       0  3577.6      .1       0
    3919     .05       0  4140.3      .1       0  4351.7     .05       0
  4457.3      .1       0  4657.6     .05       0  4756.6      .1       0
  4855.7     .05       0  5001.7     .04       0  5007.7     .05       0
  5305.6      .1       0    5614     .08       0  5976.1     .08       0
  6141.5      .1       0  6283.6      .1       0
#XS Ineff= 2 , 0
         4588.07   98.71
Permanent Ineff=
       F       F
Bank Sta=5001.7,5007.7
XS Rating Curve= 0 ,0
Exp/Cntr=0.3,0.1

Type RM Length L Ch R = 1 ,9665    ,404,404,404
BEGIN DESCRIPTION:
Mapping XS 0bbca69d
END DESCRIPTION:
XS GIS Cut Line= 4
      2305497.56     13250204.45      2305042.27     13249450.38
      2304202.86     13247807.12      2303313.65     13246981.94
#Sta/Elev= 30
  2694.3  140.34  2948.5  135.49  3135.4  120.56  3181.8  118.55  3187.6  122.78
  3193.8  117.22    3209  116.86  3224.5  126.08  3245.9  121.28  3261.4  126.16
  3427.4  120.72  3515.6  124.99  3640.5  114.51  3701.5  100.37  3970.2    92.8
  4030.9   92.66  4481.4   93.84  4530.6   91.86  4533.3   91.36  4536.6   91.86
  4610.4   92.08    4802   93.15    4816    93.2  4940.3   93.29  5029.2   93.82
  5262.3   96.87  5536.8  110.48  5754.7  116.86  5884.2   118.2  6633.5  145.11
#Mann= 11 ,-1 , 0
  2694.3      .1       0  3970.2     .05       0  4030.9      .1       0
  4481.4     .05       0  4530.6     .07       0  4536.6     .05       0
  4610.4      .1       0    4802     .05       0    4816      .1       0
  5536.8     .08       0  5754.7      .1       0
Bank Sta=4940.3,5029.2
XS Rating Curve= 0 ,0
Exp/Cntr=0.3,0.1

Type RM Length L Ch R = 1 ,9261    ,762,762,762
BEGIN DESCRIPTION:
UNT001 IN PECR 16.0
END DESCRIPTION:
XS GIS Cut Line= 2
      2305960.46     13249074.29       2303252.4     13246587.56
#Sta/Elev= 30
  3225.2  135.55  3248.1  135.24  3332.4  134.02    3580  126.76  3807.5   117.9
  3923.3  110.94  3993.9  107.06  4125.4  101.24  4279.8    94.3  4286.3   93.82
  4354.5   91.21  4357.3   90.71  4360.5   91.21  4427.1   91.21    4578   92.15
  4728.9   91.99  4805.4   92.57  4921.3   92.08  4966.7   93.61  5181.7   93.58
  5199.7   94.18  5520.5  104.78  5584.1  107.58  5744.8  116.89  5787.3  116.74
  5894.1  122.12  6247.3  130.05  6445.8  137.42  6714.7   154.6  6901.8  162.39
#Mann= 20 ,-1 , 0
  3225.2     .05       0  3248.1      .1       0  3332.4     .05       0
    3580      .1       0  3807.5     .05       0  3923.3      .1       0
  3993.9     .05       0  4125.4      .1       0  4286.3     .05       0
  4354.5     .07       0  4360.5     .05       0  4427.1     .12       0
    4578     .05       0  4728.9      .1       0  4805.4     .05       0
  4921.3     .12       0  5181.7     .05       0  5520.5      .1       0
  5584.1     .08       0  5894.1      .1       0
Bank Sta=4279.8,5199.7
XS Rating Curve= 0 ,0
Exp/Cntr=0.3,0.1
