--- UNT027 IN PECR.prj (project) ---

Proj Title=UNT027 IN PECR Base Level Engineering
Current Plan=p01
Default Exp/Contr=0.3,0.1
English Units
Geom File=g01
Flow File=f01
Plan File=p01
Y Axis Title=Elevation
X Axis Title(PF)=Main Channel Distance
X Axis Title(XS)=Station
BEGIN DESCRIPTION:
UNT027 IN PECR
END DESCRIPTION:
DSS Export Rating Curves= 0
DSS Export Rating Curve Sorted= 0
DSS Export Volume Flow Curves= 0
DXF OffsetX= 0
DXF OffsetY= 0
DXF ScaleX= 1
DXF ScaleY= 10

--- UNT027 IN PECR.p01 (plan) ---

Plan Title=Multiple Run
Short Identifier=Multiple
Geom File=g01
Flow File=f01
Subcritical Flow
K Sum by GR= 0
Std Step Tol= 0.01
Critical Tol= 0.01
Num of Std Step Trials= 20
Max Error Tol= 0.3
Flow Tol Ratio= 0.001
Split Flow NTrial= 30
Split Flow Tol= 0.02
Split Flow Ratio= 0.02
Log Output Level= 0
Friction Slope Method= 1
Unsteady Friction Slope Method= 2
Unsteady Bridges Friction Slope Method= 1
Parabolic Critical Depth
Global Vel Dist=  1 , 1 , 1
Global Log Level= 0
CheckData=True
Encroach Param= -1, 0, 0, 0
BEGIN DESCRIPTION:
Multiple Run
END DESCRIPTION:

--- UNT027 IN PECR.f01 (steady flow) ---

Flow Title=Multiple
Program Version=4.10
Number of Profiles= 7
Profile Names=10-year,25-year,50-year,1pct_min,100-year,1pct_plu,500-year
River Rch & RM=UNT027 IN PECR,Reach-1         ,34082
     190     255     308     274     370     500     541
River Rch & RM=UNT027 IN PECR,Reach-1         ,33095
     215     291     353     315     425     575     626
River Rch & RM=UNT027 IN PECR,Reach-1         ,29364
     266     364     444     399     539     729     805
River Rch & RM=UNT027 IN PECR,Reach-1         ,24048
     432     606     752     684     925    1252    1424
River Rch & RM=UNT027 IN PECR,Reach-1         ,19297
     639     909    1138    1043    1411    1908    2200
River Rch & RM=UNT027 IN PECR,Reach-1         ,7271
     781    1118    1405    1292    1747    2363    2738
Boundary for River Rch & Prof#=UNT027 IN PECR,Reach-1         , 1
Up Type= 0
Dn Type= 3
Dn Slope=0.0014
Boundary for River Rch & Prof#=UNT027 IN PECR,Reach-1         , 2
Up Type= 0
Dn Type= 3
Dn Slope=0.0014
Boundary for River Rch & Prof#=UNT027 IN PECR,Reach-1         , 3
Up Type= 0
Dn Type= 3
Dn Slope=0.0014
Boundary for River Rch & Prof#=UNT027 IN PECR,Reach-1         , 4
Up Type= 0
Dn Type= 3
Dn Slope=0.0014
Boundary for River Rch & Prof#=UNT027 IN PECR,Reach-1         , 5
Up Type= 0
Dn Type= 3
Dn Slope=0.0014
Boundary for River Rch & Prof#=UNT027 IN PECR,Reach-1         , 6
Up Type= 0
Dn Type= 3
Dn Slope=0.0014
Boundary for River Rch & Prof#=UNT027 IN PECR,Reach-1         , 7
Up Type= 0
Dn Type= 3
Dn Slope=0.0014
DSS Import GetInterval= 0
DSS Import GetPeak= 0
DSS Import FillOption= 0

--- UNT027 IN PECR.g01 (geometry) ---

Geom Title=Existing Conditions
Program Version=4.10

River Reach=UNT027 IN PECR  ,Reach-1
Reach XY= 30
      2277711.78     13199957.35       2279642.4     13200056.32
      2282636.24     13199483.73      2283184.76     13199215.85
      2283223.78     13198333.84      2284967.07     13197046.97
      2284901.49     13196624.68      2285815.98      13196623.1
      2286222.84     13196017.91      2287326.34     13196523.35
      2287734.26     13195500.07      2288676.34     13195218.02
      2289104.38     13195743.42      2289795.74     13195431.44
      2289719.14     13195100.02      2290506.71     13195191.44
      2290482.37     13195750.45      2291117.89     13195994.99
      2291515.94     13195801.17      2291294.96     13195060.41
      2292397.69     13195806.88      2293566.07      13194940.1
      2295049.11      13195018.7      2295305.88     13194276.68
      2296435.57     13193866.07      2296296.94     13193181.83
      2297490.38     13193171.37      2297241.23     13192286.39
      2297736.59     13192582.86      2298192.78     13191892.44

Type RM Length L Ch R = 1 ,34082   ,315,315,315
BEGIN DESCRIPTION:
UNT027 IN PECR 63.0
END DESCRIPTION:
XS GIS Cut Line= 3
      2278187.72     13200446.84      2278137.72     13199846.85
      2278037.72     13199546.84
#Sta/Elev= 30
  4406.5  274.37  4446.6  273.58  4464.2  271.51  4472.8  271.54  4496.8  270.99
  4506.8   269.9    4557  269.05  4584.6  267.38  4589.6   267.7  4617.2  266.02
  4657.3  264.89  4717.6  262.21  4747.7  261.57  4817.9  258.83  4825.4  259.19
    4838  257.46  4842.3  257.68  4878.1  257.49  4958.4  255.71  4978.5  253.97
  4995.5  251.02  4998.3  250.52  5001.5  251.02  5006.1  253.04  5011.2  253.04
  5029.6   255.7  5103.4  258.02    5114  257.86  5125.5  258.69  5324.8  265.31
#Mann= 6 ,-1 , 0
  4406.5     .05       0  4472.8      .1       0  4842.3     .12       0
  4995.5     .07       0  5001.5     .12       0  5125.5      .1       0
Bank Sta=4958.4,5029.6
XS Rating Curve= 0 ,0
Exp/Cntr=0.3,0.1

Type RM Length L Ch R = 1 ,33767   ,298,298,298
BEGIN DESCRIPTION:
Mapping XS 381c01b5
END DESCRIPTION:
XS GIS Cut Line= 4
      2278379.59     13200405.41      2278427.51     13200032.73
      2278443.48      13199686.7      2278310.39     13199383.25
#Sta/Elev= 30
  4388.5  271.87  4407.2   270.8    4508   267.9  4528.2  266.29  4538.3   266.3
  4566.7  264.64  4651.9  261.57  4659.3  260.99  4725.7  259.61  4759.7  257.98
  4770.1  258.51  4825.3  256.72  4890.3  255.49  4900.3  254.53  4910.3  255.11
  4930.3   253.2  4950.3  253.62  4960.3  253.08  4970.3  254.31  4990.4  250.88
  4997.4  250.68  5000.1  250.18  5003.4  250.68  5010.4  251.67  5020.4  251.96
  5030.4  254.81  5050.4  254.99  5064.5  255.94  5382.2     265    5442  267.35
#Mann= 6 ,-1 , 0
  4388.5     .05       0  4651.9      .1       0  4825.3     .12       0
  4997.4     .07       0  5003.4     .12       0  5064.5      .1       0
Bank Sta=4910.3,5030.4
XS Rating Curve= 0 ,0
Exp/Cntr=0.3,0.1

Type RM Length L Ch R = 1 ,33469   ,374,374,374
BEGIN DESCRIPTION:
UNT027 IN PECR 62.0
END DESCRIPTION:
XS GIS Cut Line= 4
       2278581.9     13200400.02      2278704.34     13200064.67
      2278720.31      13199686.7      2278487.06     13199310.33
#Sta/Elev= 30
  4480.3  268.64  4508.6   267.8  4526.3  267.43  4536.3  266.45  4566.8     266
  4602.7  264.37  4696.6  261.72  4714.3  260.64  4775.4  259.38  4845.1  256.37
  4859.5  256.46  4895.2  256.04  4915.2  254.08  4925.2  254.93  4935.2  252.43
  4945.2  251.91  4965.2  252.01  5002.3  250.12    5005  249.62  5008.3  250.12
  5015.3  251.07  5045.3  253.05  5055.3   253.7  5065.3  253.25  5095.3  254.45
  5119.7  254.56  5155.4  255.33  5289.4   256.2  5420.6  258.44  5658.4  265.12
#Mann= 6 ,-1 , 0
  4480.3     .05       0  4508.6      .1       0  4859.5     .12       0
  5002.3     .07       0  5008.3     .12       0  5119.7      .1       0
Bank Sta=4925.2,5045.3
XS Rating Curve= 0 ,0
Exp/Cntr=0.3,0.1

Type RM Length L Ch R = 1 ,33095   ,340,340,340
BEGIN DESCRIPTION:
UNT027 IN PECR 61.0
END DESCRIPTION:
XS GIS Cut Line= 4
      2278752.22     13200506.56      2278959.87     13200176.46
      2279156.84     13199601.52        2279263.     13199293.63
#Sta/Elev= 30
    4314  267.57  4338.5  266.61  4384.3  266.18  4390.3  265.25  4405.5  265.31
  4499.8  261.98  4542.2  261.41  4557.5  260.28  4563.4  260.73  4700.8  256.67
  4773.4   255.9  4879.9  253.41  4898.5  252.53  4904.4  253.04  4961.1  251.63
  4978.4  250.07  4989.4  247.33  4992.1  246.83  4995.4  247.33  5023.6  250.19
  5031.2  252.47  5054.9  253.27  5142.6  254.19  5284.9  256.68  5311.5  257.97
  5419.5  261.22  5450.7   261.3  5601.4  264.68  5606.7  264.31  5637.4  265.82
#Mann= 5 ,-1 , 0
    4314      .1       0  4879.9     .12       0  4989.4     .07       0
  4995.4     .12       0  5142.6      .1       0
Bank Sta=4961.1,5031.2
XS Rating Curve= 0 ,0
Exp/Cntr=0.3,0.1

Type RM Length L Ch R = 1 ,32755   ,541,541,541
BEGIN DESCRIPTION:
UNT027 IN PECR 60.0
END DESCRIPTION:
XS GIS Cut Line= 3
      2279287.72      13200696.9      2279337.72     13200046.85
      2279537.72     13199246.84
#Sta/Elev= 30
  4367.4  268.79  4576.2  261.96  4738.5  256.55    4889  252.98  4911.3  253.04
  4929.1  252.69  4949.2  251.01  4959.2  251.99  4969.2  250.72  4979.2  251.49
  4989.3     247  4996.3   245.7  4999.1   245.2  5002.3   245.7  5009.3  248.92
  5016.9  249.69  5042.6   249.6  5060.6  248.18  5070.9   249.9  5101.8  251.75
  5230.9  252.69  5277.1  252.93  5372.4  255.13  5496.1  258.76  5532.2  260.59
  5586.3  261.88  5738.3  267.37  5784.7  268.32  5792.4  269.15    5844  270.37
#Mann= 6 ,-1 , 0
  4367.4     .05       0  4576.2      .1       0  4911.3     .12       0
  4996.3     .07       0  5002.3     .12       0  5230.9      .1       0
Bank Sta=4979.2,5070.9
XS Rating Curve= 0 ,0
Exp/Cntr=0.3,0.1

Type RM Length L Ch R = 1 ,32214   ,386,386,386
BEGIN DESCRIPTION:
UNT027 IN PECR 59.0
END DESCRIPTION:
XS GIS Cut Line= 3
      2279854.22     13200666.18       2279827.6     13200224.37
      2279742.58      13199326.3
#Sta/Elev= 30
  4304.3  266.86  4413.8  264.17  4544.1  259.36  4554.1   259.5  4644.2  256.17
  4674.3  255.78  4704.4  254.17  4746.9  253.67  4754.5  252.73  4837.2  251.53
  4965.4  249.46  4985.5  248.34  4995.5  247.11  5007.7  243.01  5010.5  242.51
  5013.7  243.01  5015.8  245.21  5025.7  247.34  5035.7  246.11  5055.8  248.82
  5085.9  250.28    5096  249.92  5108.9  250.43  5227.3  253.11  5256.7  254.55
  5266.7  254.07  5337.1  255.97  5497.8  263.08  5537.2  264.01    5649   268.5
#Mann= 5 ,-1 , 0
  4304.3      .1       0  4837.2     .12       0  5007.7     .07       0
  5013.7     .12       0  5108.9      .1       0
Bank Sta=4985.5,5055.8
XS Rating Curve= 0 ,0
Exp/Cntr=0.3,0.1

Type RM Length L Ch R = 1 ,31828   ,399,399,399
BEGIN DESCRIPTION:
UNT027 IN PECR 58.0
END DESCRIPTION:
XS GIS Cut Line= 3
      2280157.66     13200533.12      2280168.31     13200213.73
      2280083.13      13199372.6
#Sta/Elev= 30
  4442.5   265.8  4488.8  264.87  4498.8  263.81  4548.8  261.76  4738.9  255.73
  4799.1  252.99  4820.9  253.25    4833  252.64  4879.5   250.6  4899.6  250.48
  4915.8   248.7  4920.8  249.02  4939.8   248.2  4949.9   248.6  4959.9  247.25
    4970  245.27  4997.2  242.82  4999.9  242.32  5003.2  242.82  5015.6  246.06
  5020.7  245.96  5030.3  247.76  5123.9  248.21  5150.9  248.16    5171  249.29
  5241.4  251.54  5251.4  251.38    5372  255.97  5382.1  256.98  5607.5  265.16
#Mann= 5 ,-1 , 0
  4442.5      .1       0    4833     .12       0  4997.2     .07       0
  5003.2     .12       0  5123.9      .1       0
Bank Sta=4959.9,5030.3
XS Rating Curve= 0 ,0
Exp/Cntr=0.3,0.1

Type RM Length L Ch R = 1 ,31429   ,447,447,447
BEGIN DESCRIPTION:
UNT027 IN PECR 57.0
END DESCRIPTION:
XS GIS Cut Line= 3
      2280587.73      13200496.9      2280437.72     13199796.85
      2280337.73      13199396.9
#Sta/Elev= 30
  4295.4  267.63    4315  267.61  4320.2   266.8  4346.6  265.65  4369.6  265.31
  4448.9  261.75  4489.8  260.97  4512.8  259.26  4613.1  255.62  4663.6  253.55
  4735.2  251.72  4744.6  250.81    4807   249.6  4837.5  248.34    4950  246.71
  4960.2  244.23  4980.7  243.26  4986.6  241.91  4991.7  242.04  4998.1  240.32
  5000.9  239.82  5004.1  240.32  5008.8  243.13  5013.9  243.13  5021.6  245.09
  5029.4  246.49  5053.8  247.49  5186.6   251.8  5382.4  260.42  5423.6  261.33
#Mann= 6 ,-1 , 0
  4295.4     .05       0  4613.1      .1       0    4807     .12       0
  4998.1     .07       0  5004.1     .12       0  5053.8      .1       0
Bank Sta=4960.2,5021.6
XS Rating Curve= 0 ,0
Exp/Cntr=0.3,0.1

Type RM Length L Ch R = 1 ,30982   ,497,497,497
BEGIN DESCRIPTION:
UNT027 IN PECR 56.0
END DESCRIPTION:
XS GIS Cut Line= 4
      2280924.25     13200474.58      2280908.28     13199952.87
      2280801.81     13199473.75      2280556.92     13199186.27
#Sta/Elev= 30
  4281.9  266.14  4339.6  264.72  4389.7  262.28  4399.7  262.44  4407.4  261.47
  4656.8  252.82  4769.8  249.94  4846.7  247.05    4871  245.67  4902.2  245.68
  4919.6  244.11  4924.7  244.25  4932.9  242.81  4943.2  242.54  4953.4  244.22
  4963.2  244.82  4973.9  243.06  4984.2  240.39  5001.6  238.14  5004.4  237.64
  5007.6  238.14  5011.8  241.29  5016.9  241.29  5025.1  244.28  5045.6  245.44
  5103.7  245.65    5189  246.96  5288.4  249.68  5609.9   261.1  5672.3  262.87
#Mann= 7 ,-1 , 0
  4281.9     .05       0  4407.4      .1       0  4846.7     .12       0
  5001.6     .07       0  5007.6     .12       0  5103.7      .1       0
  5609.9     .05       0
Bank Sta=4973.9,5025.1
XS Rating Curve= 0 ,0
Exp/Cntr=0.3,0.1

Type RM Length L Ch R = 1 ,30485   ,544,544,544
BEGIN DESCRIPTION:
UNT027 IN PECR 55.0
END DESCRIPTION:
XS GIS Cut Line= 3
      2281209.66     13200493.74      2281327.73     13199847.86
      2281265.23     13198972.87
#Sta/Elev= 30
  4192.1  261.84  4239.8  260.23  4524.4   253.9  4594.4  251.47  4676.9   249.9
    4687  248.95  4839.4   245.7  4916.9  244.42    4970  240.99    4980  239.98
    4990  240.14  5000.1  237.39  5007.1  236.86  5009.8  236.36  5013.1  236.86
  5020.1  239.63  5030.1  240.85  5040.2  242.16  5050.2  242.09  5062.3  243.42
  5242.6  245.25  5250.7  245.95  5270.8  245.45  5290.8  246.04  5310.9  247.09
  5471.3  251.67  5491.3  252.84  5511.4  253.06  5551.5  255.14  5725.9  260.15
#Mann= 5 ,-1 , 0
  4192.1      .1       0  4839.4     .12       0  5007.1     .07       0
  5013.1     .12       0  5242.6      .1       0
Bank Sta=4970,5030.1
XS Rating Curve= 0 ,0
Exp/Cntr=0.3,0.1

Type RM Length L Ch R = 1 ,29941   ,498,498,498
BEGIN DESCRIPTION:
UNT027 IN PECR 54.0
END DESCRIPTION:
XS GIS Cut Line= 3
      2281848.57     13200375.67      2281671.48     13199469.39
      2281480.53     13199087.49
#Sta/Elev= 30
  3968.9  258.31    4039   256.1  4052.9  256.45  4059.4  255.58  4207.5  251.46
  4315.7  249.41  4385.4  246.98  4418.8  246.99  4644.7  243.78  4721.7  242.72
  4733.2  243.25  4813.4  241.55  4848.7   241.5  4861.7  241.48  4956.6  240.73
  4962.2  238.57  4984.6  237.14  5001.1  235.35    5007  236.51  5040.5  239.29
  5068.4  242.66    5074  244.61  5085.2  246.41  5107.6  246.84  5135.5  248.49
  5230.6  252.94  5247.3   253.2  5252.9  254.21  5286.5  254.79  5319.3  256.44
#Mann= 7 ,-1 , 0
  3968.9      .1       0  4644.7     .12       0  4848.7      .1       0
  4861.7     .12       0  4962.2     .07       0  5040.5     .12       0
  5135.5      .1       0
Bank Sta=4962.2,5040.5
XS Rating Curve= 0 ,0
Exp/Cntr=0.3,0.1

Type RM Length L Ch R = 1 ,29443   ,79,79,79
BEGIN DESCRIPTION:
UNT027 IN PECR 53.0
END DESCRIPTION:
XS GIS Cut Line= 3
      2282341.62     13200136.07      2282282.59      13199830.5
      2281775.66     13199031.92
#Sta/Elev= 30
  4252.7  247.45  4328.5  246.06  4593.7  242.43  4671.1  241.69  4852.5  240.54
  4947.3  237.84  4996.7  236.59  5027.2  236.78  5032.9  235.92    5042  237.28
  5063.6  237.77  5338.1  245.46  5345.7  246.65  5351.6  245.92  5382.1  247.75
  5388.1   247.5  5403.3  248.84  5409.2  248.35  5418.6  249.14  5424.5  248.53
  5432.9  249.29  5439.7  250.89  5445.7  249.48  5460.9  250.19  5476.2  252.29
  5482.1  251.22  5491.4  252.56  5497.3  251.37  5503.9  252.78  5509.8  252.78
#Mann= 7 ,-1 , 0
  4252.7      .1       0  4328.5     .08       0  4593.7      .1       0
  4671.1     .12       0  4947.3     .08       0  4947.3     .07       0
  5063.6     .12       0
Bank Sta=4947.3,5063.6
XS Rating Curve= 0 ,0
Exp/Cntr=0.3,0.1

Type RM Length L Ch R = 1 ,29364   ,143,143,143
BEGIN DESCRIPTION:
UNT027 IN PECR 52.0
END DESCRIPTION:
XS GIS Cut Line= 3
      2282442.32     13200129.15      2282352.03     13199795.78
      2281832.75     13198971.85
#Sta/Elev= 30
  4220.5  245.79  4390.7  243.86  4521.1  241.73  4576.4  242.53  4588.8   240.5
  4601.9  240.65  4655.8  239.31  4718.4  240.16  4728.8  238.83  4741.9  240.61
    4750  238.88  4771.2  240.26    4840  238.69  4850.1  239.79  4859.4  238.23
  4865.4   239.8  4880.6  237.74    4996  236.67  5032.2  234.99  5074.9  236.63
  5126.7  236.68    5242  240.43  5257.3  242.22  5278.5  241.53  5293.8  245.25
  5299.7  243.26  5309.1  246.23    5315  245.23  5330.3  247.23  5539.8  255.01
#Mann= 8 ,-1 , 0
  4220.5     .08       0  4390.7     .05       0  4521.1     .08       0
  4601.9     .05       0  4718.4     .08       0    4840     .12       0
    4996     .07       0  5074.9     .12       0
Bank Sta=4996,5074.9
XS Rating Curve= 0 ,0
Exp/Cntr=0.3,0.1

Type RM Length L Ch R = 1 ,29221   ,556,556,556
BEGIN DESCRIPTION:
Mapping XS d0a25309
END DESCRIPTION:
XS GIS Cut Line= 4
      2282472.49     13200099.79      2282302.35     13199551.15
      2282215.54     13199398.38       2281906.5     13198946.96
#Sta/Elev= 30
  4154.3  245.57  4210.7  244.83  4294.5  243.82  4521.7  241.71    4527  240.52
  4554.3  241.68  4559.6  240.87  4662.5  240.12  4690.6   238.8  4818.8  238.08
  4918.4  237.54  4931.8  235.07  4946.8  233.12  4967.7  235.29  4976.6  233.55
  5003.6  233.24  5012.2  232.04  5018.5  232.76  5027.4  239.78  5048.3  238.55
  5054.4  235.97  5063.3  236.52  5069.3  235.83  5084.2  238.13  5090.3   236.8
  5112.3  238.16  5120.1  241.98  5191.9  243.63  5227.7  245.68  5451.5  253.89
#Mann= 7 ,-1 , 0
  4154.3     .05       0  4210.7     .08       0  4294.5     .05       0
  4690.6     .12       0  4818.8     .05       0  4931.8     .04       0
  5027.4     .05       0
Bank Sta=4931.8,5027.4
XS Rating Curve= 0 ,0
Exp/Cntr=0.3,0.1

Type RM Length L Ch R = 1 ,28665   ,273,273,273
BEGIN DESCRIPTION:
UNT027 IN PECR 51.0
END DESCRIPTION:
XS GIS Cut Line= 4
      2282805.82     13200058.11      2282687.76     13199596.29
      2282552.35     13199262.96      2282317.01     13198930.72
#Sta/Elev= 30
  4398.6  247.24  4482.9  245.24  4612.2  242.16  4653.1  241.87  4668.3  241.08
  4864.4  238.68  4930.8  238.41    4961  237.78  4972.8   236.3  4982.6  234.21
  4991.5  230.08  4993.9  229.86  4996.6  229.36  4999.9  229.86    5003   229.9
    5015  231.28  5026.3  231.47  5036.6  232.57    5045  234.55  5050.4  235.44
  5074.5  234.68  5090.5  235.35  5110.9  235.15  5133.7  236.06  5152.1  235.96
  5229.8  236.69  5279.3  237.52  5285.9   238.1  5487.6  238.91  5642.2  242.45
#Mann= 8 ,-1 , 0
  4398.6     .05       0  4482.9      .1       0  4930.8     .12       0
  4993.9     .07       0  4999.9     .12       0    5003      .1       0
  5110.9     .12       0  5152.1      .1       0
Bank Sta=4982.6,5045
XS Rating Curve= 0 ,0
Exp/Cntr=0.3,0.1

Type RM Length L Ch R = 1 ,28392   ,623,623,623
BEGIN DESCRIPTION:
UNT027 IN PECR 50.0
END DESCRIPTION:
XS GIS Cut Line= 4
      2283156.51     13199950.45      2282975.96     13199565.04
      2282784.99     13199196.99      2282438.22     13198881.43
#Sta/Elev= 30
    4304  248.64  4462.6  243.57  4610.3  240.45  4695.5  238.78  4734.5  238.33
  4795.2  237.25    4862  234.93  4889.8  235.28  4964.8  233.84  4978.3  233.73
  4986.7  230.19  4997.4  228.29  5000.1  227.79  5003.4  228.29  5006.4  229.46
  5009.2  230.55  5016.9  230.28  5022.5  231.25    5039  232.11  5044.6  233.95
  5076.8  234.25  5141.5  237.04  5192.2  237.96  5198.9   237.3  5213.8  237.71
  5255.7  238.37    5355  236.89  5461.1   237.5  5602.3  239.46  5613.1  240.41
#Mann= 9 ,-1 , 0
    4304      .1       0  4610.3     .12       0  4695.5      .1       0
  4734.5     .12       0  4964.8     .16       0  4997.4     .07       0
  5003.4     .16       0  5006.4     .12       0  5213.8      .1       0
Bank Sta=4978.3,5044.6
XS Rating Curve= 0 ,0
Exp/Cntr=0.3,0.1

Type RM Length L Ch R = 1 ,27769   ,475,475,475
BEGIN DESCRIPTION:
UNT027 IN PECR 49.0
END DESCRIPTION:
XS GIS Cut Line= 4
      2283583.57     13199037.26      2283347.49     13198992.13
      2282819.71     13198964.35      2282538.47     13198804.63
#Sta/Elev= 30
  4567.3  244.38  4609.8  243.26  4784.7  238.85  4802.2  238.33  4867.5  236.33
  4947.6  232.16  4957.6   229.1  4967.6  228.33  4987.7  228.78  4994.7  227.51
  4997.4  227.01  5000.7  227.51  5007.9  227.55  5017.7  228.78  5027.7  229.11
  5037.7  228.17  5047.8  228.68  5067.8  231.34  5077.8  231.05  5087.8  231.83
  5117.9  232.14  5147.9  234.26  5167.9  234.06    5188  234.88  5198.2  234.63
  5288.1   236.2  5379.5  236.17  5423.5  235.74  5498.5  236.08  5659.6  238.69
#Mann= 7 ,-1 , 0
  4567.3      .1       0  4609.8     .05       0  4784.7      .1       0
  4802.2     .12       0  4994.7     .07       0  5000.7     .12       0
  5379.5      .1       0
Bank Sta=4947.6,5067.8
XS Rating Curve= 0 ,0
Exp/Cntr=0.3,0.1

Type RM Length L Ch R = 1 ,27294   ,386,386,386
BEGIN DESCRIPTION:
UNT027 IN PECR 48.0
END DESCRIPTION:
XS GIS Cut Line= 3
      2283552.39     13198728.26       2283295.4     13198585.88
      2282761.71     13198447.25
#Sta/Elev= 30
  4542.1  241.43    4560  241.27    4592  239.57  4787.4  232.32  4838.3  231.13
  4850.4  231.09  4855.6  230.46  4936.8  228.57  4972.1  228.75  4988.5  227.91
  4995.8   224.4  4998.6   223.9  5001.8   224.4  5007.5  225.86  5019.5   225.3
  5029.8  226.78  5040.1  228.44  5060.8  228.65  5088.6  230.29  5127.8  231.02
  5143.5   231.6  5169.7  231.77  5174.9   232.7  5184.8  232.14  5205.1  232.42
  5215.8   233.6  5236.4  234.49  5250.8     234  5277.8  235.47  5387.3  238.35
#Mann= 6 ,-1 , 0
  4542.1      .1       0  4787.4     .16       0  4838.3     .12       0
  4995.8     .07       0  5001.8     .12       0  5127.8      .1       0
Bank Sta=4988.5,5029.8
XS Rating Curve= 0 ,0
Exp/Cntr=0.3,0.1

Type RM Length L Ch R = 1 ,26908   ,138,138,138
BEGIN DESCRIPTION:
UNT027 IN PECR 47.0
END DESCRIPTION:
XS GIS Cut Line= 3
      2283737.69     13198596.83      2283337.72     13198246.85
      2283087.73     13198096.86
#Sta/Elev= 30
  4485.9  245.97  4670.5   237.2  4719.8  235.42  4742.2  233.94  4861.2  228.52
  4883.1  228.44  4889.7  231.34  4897.3  232.78  4903.9  233.11  4911.1  232.93
  4919.5  230.94  4939.1  227.28  4953.3  224.62  4975.1  223.46  4981.8  222.49
  5003.6  222.23  5007.2  221.08    5010  220.58  5013.2  221.08  5040.7  222.01
  5067.9  226.98  5075.7  227.77  5083.5  230.72  5089.3  234.36    5099  234.68
  5110.7  233.56  5126.2  230.62  5194.4   233.5  5205.9  234.45  5308.9  238.41
#Mann= 6 ,-1 , 0
  4485.9     .05       0  4742.2     .16       0  4919.5     .12       0
  5007.2     .07       0  5013.2     .12       0  5194.4      .1       0
Bank Sta=4939.1,5067.9
XS Rating Curve= 0 ,0
Exp/Cntr=0.3,0.1

Type RM Length L Ch R = 1 ,26770   ,320,320,320
BEGIN DESCRIPTION:
Mapping XS 4af06c68
END DESCRIPTION:
XS GIS Cut Line= 4
      2283826.68     13198568.54      2283496.79     13198231.71
      2283441.24     13198148.38       2283146.1     13197936.57
#Sta/Elev= 30
  4485.1   248.5  4655.3  240.98  4782.5  234.44    4802  232.86  4895.7  228.33
  4916.9  229.02  4923.9  227.52  4931.1     227  4938.1  230.24  4945.2  229.52
  4952.2  230.57  4960.2  230.45  4966.2  228.42  4974.4  228.91  4987.2  226.34
  4996.2  224.18  5007.5  223.35  5010.2  222.85  5013.5  223.35  5017.2  224.97
  5023.3  225.22  5032.3  229.97  5038.3  226.39  5046.5   230.2  5053.3   231.2
  5082.3  231.34  5089.6  230.12  5103.2  229.62  5275.1  234.44    5420  240.11
#Mann= 5 ,-1 , 0
  4485.1     .05       0    4802     .16       0  5007.5     .07       0
  5013.5     .16       0  5089.6      .1       0
Bank Sta=4987.2,5032.3
XS Rating Curve= 0 ,0
Exp/Cntr=0.3,0.1

Type RM Length L Ch R = 1 ,26450   ,453,453,453
BEGIN DESCRIPTION:
UNT027 IN PECR 46.0
END DESCRIPTION:
XS GIS Cut Line= 3
      2283837.71     13198296.84      2283737.72     13198046.85
      2283337.74     13197646.87
#Sta/Elev= 30
  4732.3  239.15  4747.1  238.01  4776.7  236.98  4807.7  234.91  4818.4  234.65
  4825.2  233.81    4840  233.37  4877.9  230.75  4903.3  229.09  4915.4  228.83
  4947.7  226.56    4980  225.51  4986.7  224.15  4992.1  222.03  4995.9  221.46
  4998.6  220.96  5001.9  221.46  5015.7  222.16  5029.8  223.42    5044  223.25
  5052.5  222.69  5058.1  222.32  5086.4  225.11  5171.2  229.23  5284.4  231.75
    5341  232.41  5411.7  234.32  5489.5  237.32  5553.1  239.83  5567.2  240.76
#Mann= 6 ,-1 , 0
  4732.3     .05       0  4877.9     .12       0  4995.9     .07       0
  5001.9     .12       0  5052.5      .1       0  5489.5     .05       0
Bank Sta=4980,5086.4
XS Rating Curve= 0 ,0
Exp/Cntr=0.3,0.1

Type RM Length L Ch R = 1 ,25997   ,178,178,178
BEGIN DESCRIPTION:
UNT027 IN PECR 45.0
END DESCRIPTION:
XS GIS Cut Line= 3
       2284237.7     13198046.82      2284037.72     13197746.85
      2283637.74     13197396.87
#Sta/Elev= 30
  4645.3  237.83  4667.8  237.31  4681.3  236.29  4724.9  234.73  4739.9  234.62
  4789.5  232.11    4797  232.47    4818   230.7  4848.1  229.62  4900.6  226.51
  4920.2  225.81  4947.2  223.91  4956.2  223.04  4962.2  221.69  4992.3  220.44
  4995.3  218.84  4998.1  218.34  5001.3  218.84  5002.8  220.15  5009.1  220.15
  5019.6  221.57  5084.1  223.81  5112.1  224.26  5175.9  226.59    5311  230.06
  5324.7   229.9  5338.5  230.77  5388.8  231.62  5481.1  234.81  5537.3  236.68
#Mann= 6 ,-1 , 0
  4645.3     .05       0  4900.6     .12       0  4995.3     .07       0
  5001.3     .12       0  5175.9      .1       0  5481.1     .05       0
Bank Sta=4947.2,5084.1
XS Rating Curve= 0 ,0
Exp/Cntr=0.3,0.1

Type RM Length L Ch R = 1 ,25819   ,125,125,125
BEGIN DESCRIPTION:
Mapping XS fab47697
END DESCRIPTION:
XS GIS Cut Line= 2
      2284497.86      13197955.5      2283806.91     13197268.02
#Sta/Elev= 30
  4536.4   234.7  4691.1  232.83  4712.3  231.79  4818.4  229.17  4912.8  225.46
  4938.6  224.01  4952.7  222.66  4959.8  220.63    4981  218.27  4988.1  217.01
  4999.2  216.42    5002  215.92  5005.2  216.42  5030.5  217.53  5037.6  219.55
  5058.8  222.69  5065.9  224.49  5072.9  225.47    5080  225.33  5087.1  224.48
  5094.2   222.6  5111.8  222.84  5143.6  223.92  5193.2  225.38  5207.3   226.5
  5270.9  228.23  5285.1  228.96  5299.2  228.96  5368.1  230.79  5511.1  233.65
#Mann= 6 ,-1 , 0
  4536.4     .05       0  4912.8     .12       0  4999.2     .07       0
  5005.2     .12       0  5111.8      .1       0  5368.1     .05       0
Bank Sta=4938.6,5143.6
XS Rating Curve= 0 ,0
Exp/Cntr=0.3,0.1

Type RM Length L Ch R = 1 ,25694   ,76,76,76
BEGIN DESCRIPTION:
UNT027 IN PECR 44.0
END DESCRIPTION:
XS GIS Cut Line= 3
      2284543.01     13197934.67        2284293.     13197566.61
       2283852.4     13197223.15
#Sta/Elev= 30
  4503.1  233.38  4576.9  233.03  4591.9  232.18  4612.9  232.68  4878.5  225.18
  4923.6  223.32  4936.2  224.81    4948  224.91  4952.1  226.04  4958.4   224.6
  4966.6  225.56  4972.9  223.93  4980.1  225.64  4993.7  224.56  5016.3  226.01
  5022.7   224.8  5030.8  226.43  5037.1  224.39  5043.5   225.6  5051.6  225.63
  5062.3  223.48  5069.4  221.65  5072.2  221.15  5075.4  221.65  5115.8  223.21
  5130.3  224.64  5157.6  223.99  5217.2  226.95  5343.8  230.35  5506.7  232.95
#Mann= 6 ,-1 , 0
  4503.1     .05       0  4878.5     .12       0  5062.3      .1       0
  5069.4     .07       0  5075.4      .1       0  5217.2     .05       0
Bank Sta=5062.3,5115.8
XS Rating Curve= 0 ,0
Exp/Cntr=0.3,0.1

Type RM Length L Ch R = 1 ,25618   ,297,297,297
BEGIN DESCRIPTION:
Mapping XS 7f880980
END DESCRIPTION:
XS GIS Cut Line= 3
      2284577.73     13197927.73      2284386.75     13197538.83
      2283891.45     13197178.61
#Sta/Elev= 30
  4460.4  232.55  4483.7  232.03  4514.3  232.41  4542.4  231.56  4550.5   231.9
  4559.3  230.97  4617.3   230.5  4649.2  229.27  4739.2   227.6  4834.7  224.35
  4840.2   224.6  4877.1  222.89  4937.6  221.27  4966.7  221.33  4987.9  218.44
  5013.1  218.04  5015.9  217.54  5019.1  218.04  5044.3  221.13    5058  221.41
  5073.6  221.54  5088.3  222.68  5138.6   224.4  5144.7  225.47  5160.8  225.59
  5201.6  227.22  5238.7   227.6  5301.6  229.27  5424.2  231.58  5506.1  232.31
#Mann= 6 ,-1 , 0
  4460.4     .05       0  4877.1     .12       0  5013.1     .07       0
  5019.1     .12       0    5058      .1       0  5160.8     .05       0
Bank Sta=4937.6,5058
XS Rating Curve= 0 ,0
Exp/Cntr=0.3,0.1

Type RM Length L Ch R = 1 ,25321   ,568,568,568
BEGIN DESCRIPTION:
UNT027 IN PECR 43.0
END DESCRIPTION:
XS GIS Cut Line= 4
      2285002.93     13197668.68      2284759.54     13197440.04
        2284349.     13197174.54       2284032.3     13197147.54
#Sta/Elev= 30
  4391.6  234.39  4630.2  226.54  4644.4  226.86  4658.5  225.49  4747.4  222.66
  4773.4  222.15  4779.4  224.61  4800.5     226  4809.7  225.74  4815.6  222.92
  4822.1  222.23  4836.8  220.34  4888.2  218.73  4909.3  218.28  4945.6  219.44
  4960.8   219.2    4997   217.7    5000  216.65  5002.7  216.15    5006  216.65
  5012.2   217.1  5018.2  220.31  5061.2  222.92  5098.8  224.21  5148.8  225.63
  5184.4  225.02  5192.2  225.77  5248.5  225.46  5299.6  226.42  5532.3  229.39
#Mann= 8 ,-1 , 0
  4391.6     .05       0  4747.4      .1       0  4822.1     .12       0
    5000     .07       0    5006     .12       0  5098.8     .05       0
  5148.8      .1       0  5299.6     .05       0
Bank Sta=4888.2,5018.2
XS Rating Curve= 0 ,0
Exp/Cntr=0.3,0.1

Type RM Length L Ch R = 1 ,24753   ,179,179,179
BEGIN DESCRIPTION:
Mapping XS ff6e9015
END DESCRIPTION:
XS GIS Cut Line= 4
      2285132.21     13197353.25      2285059.29     13197071.99
      2285028.04      13196995.6      2284390.94       13197051.
#Sta/Elev= 30
  4584.8  231.31  4764.6  225.23  4787.7  223.92  4858.3  222.63  4867.5  221.92
  4918.9  219.99  4924.3  218.29  4942.9  217.52  4948.3  215.78  4960.6  215.27
  4968.3  213.16  4985.3  212.33  4988.1  211.83  4991.3  212.33  5018.4  212.45
  5038.5  213.35  5058.6  216.94  5068.6  219.34  5078.7  220.06  5088.7  222.09
  5098.7  222.45    5116  218.46  5118.8  217.66  5138.9   217.5    5169  218.48
  5184.4  218.87  5309.5  220.83  5319.6  221.71  5348.4  221.64  5597.4  224.69
#Mann= 8 ,-1 , 0
  4584.8     .05       0  4764.6     .12       0  4867.5     .16       0
  4985.3     .07       0  4991.3     .16       0    5116     .16       0
  5184.4      .1       0  5348.4     .05       0
Bank Sta=4924.3,5169
XS Rating Curve= 0 ,0
Exp/Cntr=0.3,0.1

Type RM Length L Ch R = 1 ,24574   ,178,178,178
BEGIN DESCRIPTION:
UNT027 IN PECR 42.0
END DESCRIPTION:
XS GIS Cut Line= 6
      2285239.86     13197308.13      2285066.24     13196835.88
      2285038.46     13196804.63      2284944.71      13196832.4
      2284903.04     13196877.54      2284378.73     13197012.96
#Sta/Elev= 30
  4370.1  231.63    4563  224.56  4726.6  219.78  4782.5  218.15  4839.9   218.7
  4895.2  221.56  4920.5  221.61  4938.4  220.43  4952.8  220.36  4970.4  219.52
  4991.3  220.85  5014.3  220.93  5023.2  220.33  5037.3  221.26  5051.5  220.56
  5076.7   220.9  5082.2  217.99  5087.6  216.84  5090.4  216.34  5093.6  216.84
  5095.8  217.39  5177.2  217.73  5206.1  218.22  5293.9  219.98  5299.1  220.78
  5323.8  221.34    5370  222.54  5410.7  222.36  5433.3  223.08  5618.2  224.76
#Mann= 7 ,-1 , 0
  4370.1     .05       0  4726.6     .16       0  4952.8     .12       0
  5087.6     .07       0  5093.6     .12       0  5177.2      .1       0
  5323.8     .05       0
Bank Sta=5082.2,5206.1
XS Rating Curve= 0 ,0
Exp/Cntr=0.3,0.1

Type RM Length L Ch R = 1 ,24396   ,348,348,348
BEGIN DESCRIPTION:
Mapping XS cff1edc0
END DESCRIPTION:
XS GIS Cut Line= 4
      2285281.52     13197294.22       2285083.6     13196710.88
      2284871.79     13196710.88      2284416.92     13196974.77
#Sta/Elev= 30
  4119.8  231.65  4333.7  223.54  4528.9  217.92  4552.6   217.5  4659.9  216.83
  4687.3  217.08  4705.3  215.75  4710.5  216.58  4735.3  215.57  4741.8  216.87
  4751.7  215.52  4784.1  216.02  4891.7  217.51  4901.7  216.69  4963.8  216.31
  4985.3  215.64  4991.1  214.74  4995.6  212.31  4998.3  211.81  5001.6  212.31
  5012.6     213  5018.7  214.96  5021.7  215.93  5034.2  216.58  5087.2  218.25
  5226.3  222.58  5305.8  223.51  5349.6     224  5371.2  223.38  5473.5  224.52
#Mann= 9 ,-1 , 0
  4119.8     .05       0  4552.6      .1       0  4659.9     .16       0
  4741.8      .1       0  4784.1     .16       0  4995.6     .07       0
  5001.6     .16       0  5018.7      .1       0  5305.8     .05       0
Bank Sta=4528.9,5087.2
XS Rating Curve= 0 ,0
Exp/Cntr=0.3,0.1

Type RM Length L Ch R = 1 ,24048   ,279,279,279
BEGIN DESCRIPTION:
UNT027 IN PECR 41.0
END DESCRIPTION:
XS GIS Cut Line= 3
      2285337.73      13197396.9      2285081.91      13196554.9
      2284937.72     13196296.85
#Sta/Elev= 30
    4120  234.94    4235  231.66  4551.9  220.22  4654.4  217.66  4683.4  217.01
  4759.6  215.97  4776.9  216.54  4830.7  216.49  4858.2  215.22  4891.1  216.14
    4924  214.17  4956.2   214.3  4967.3  215.62  4987.5  215.01    4995  211.34
  4995.6   210.1  4998.4   209.6  5001.6   210.1  5012.1   212.7  5016.9  213.72
  5022.6  213.69  5038.6  215.53  5044.3  215.08  5076.3  217.31    5098  219.04
  5103.7  218.24  5112.3  220.16  5125.4  219.58  5135.7  220.87  5295.6  227.32
#Mann= 7 ,-1 , 0
    4120     .05       0  4654.4      .1       0  4776.9     .16       0
  4995.6     .07       0  5001.6     .16       0  5012.1     .12       0
  5135.7     .05       0
Bank Sta=4683.4,5076.3
XS Rating Curve= 0 ,0
Exp/Cntr=0.3,0.1

Type RM Length L Ch R = 1 ,23769   ,487,487,487
BEGIN DESCRIPTION:
UNT027 IN PECR 40.0
END DESCRIPTION:
XS GIS Cut Line= 3
      2285553.16     13197169.66      2285490.67      13196862.4
      2285142.36      13196082.6
#Sta/Elev= 30
  4356.7  229.81  4369.8  228.96  4516.3  225.44    4655  222.35  4720.1  220.25
  4769.6  217.62  4812.8   215.6    4836  214.13  4878.6  213.61  4911.1  213.87
  4950.1  213.15  4957.5  211.58    4972  212.83  4980.7  210.98  4986.2  212.03
  4990.9  208.61  4993.7  208.11  4996.9  208.61  5004.2  209.67  5009.4  208.69
  5015.8  214.03  5070.6  215.43  5092.5  216.84  5158.1  218.22  5298.9  221.02
  5344.4  223.79  5356.3  223.79  5366.3  224.92  5433.4  227.44  5524.3  231.48
#Mann= 10 ,-1 , 0
  4356.7     .05       0  4516.3      .1       0    4655     .05       0
  4769.6      .1       0  4878.6     .16       0  4990.9     .07       0
  4996.9     .16       0  5004.2     .12       0  5158.1      .1       0
  5433.4     .05       0
Bank Sta=4812.8,5070.6
XS Rating Curve= 0 ,0
Exp/Cntr=0.3,0.1

Type RM Length L Ch R = 1 ,23282   ,527,527,527
BEGIN DESCRIPTION:
UNT027 IN PECR 39.0
END DESCRIPTION:
XS GIS Cut Line= 3
      2285922.95     13197127.98      2285870.87     13196711.36
      2285485.46     13195815.52
#Sta/Elev= 30
  4473.7  226.54  4726.8  221.45  4886.8  220.12  4952.9  219.15  4961.6  218.37
  4974.7  214.32  4985.1   211.6  4990.6  212.14  4993.4  208.52  4996.2  208.02
  4999.4  208.52  5007.3  209.67  5014.1  209.45  5019.5  211.78  5061.6   212.1
  5201.6  211.77  5399.8  214.19  5540.8  217.67  5589.7   220.4  5622.5  224.05
  5638.7  224.26  5646.1   225.7  5655.1  225.07  5669.6  226.89  5675.1  226.46
  5714.9  229.11  5767.6  230.61  5772.1  230.38  5821.7  232.97  5868.8  233.97
#Mann= 9 ,-1 , 0
  4473.7     .05       0  4886.8      .1       0  4993.4     .07       0
  4999.4      .1       0  5061.6     .12       0  5201.6      .1       0
  5655.1     .05       0  5767.6      .1       0  5772.1     .05       0
Bank Sta=4974.7,5399.8
XS Rating Curve= 0 ,0
Exp/Cntr=0.3,0.1

Type RM Length L Ch R = 1 ,22755   ,684,684,684
BEGIN DESCRIPTION:
UNT027 IN PECR 38.0
END DESCRIPTION:
XS GIS Cut Line= 5
      2286271.91     13197122.79      2286240.67     13196742.61
      2286141.71     13196383.23      2285876.08     13196138.44
      2285881.29     13195867.63
#Sta/Elev= 30
    4102  226.03  4278.5  222.92  4411.7  219.04  4579.5  214.92  4759.1  213.01
  4800.6  213.34  4849.8  212.14  4915.6  211.87  4976.8  210.95  4990.9  208.07
  4994.7  205.97  4997.5  205.47  5000.7  205.97  5005.1  207.72  5011.9  208.81
  5033.5   211.1  5045.6  211.24  5068.6  211.45  5101.5  209.21  5111.2  210.53
  5175.5   211.7  5220.7  212.77    5229  213.81    5279   217.9    5289   218.1
    5329  222.13    5339  224.84    5359  226.38  5469.1  229.85  5488.3  229.38
#Mann= 9 ,-1 , 0
    4102     .05       0  4411.7      .1       0  4579.5     .05       0
  4915.6     .12       0  4994.7     .07       0  5000.7     .12       0
  5045.6     .16       0  5101.5     .12       0  5175.5      .1       0
Bank Sta=4759.1,5229
XS Rating Curve= 0 ,0
Exp/Cntr=0.3,0.1

Type RM Length L Ch R = 1 ,22071   ,352,352,352
BEGIN DESCRIPTION:
UNT027 IN PECR 37.0
END DESCRIPTION:
XS GIS Cut Line= 3
      2286532.33     13197039.48      2286391.71      13196362.4
      2286360.46     13195742.62
#Sta/Elev= 30
  4030.2  220.26  4078.2  218.63  4228.5  218.12  4318.6  216.32  4339.3  216.59
  4349.5  218.18  4359.7  217.97  4373.8  215.73  4390.4  214.82  4451.8  214.05
  4664.3  211.85    4707   210.8  4787.4  209.73  4807.4  210.31  4817.4  209.59
  4878.1  208.97  4987.6  208.41  4994.6  205.77  4997.4  205.27  5000.6  205.77
  5052.9  209.38  5067.7  211.18  5095.8   213.4  5100.8  212.51  5107.8  214.52
  5137.8  215.98  5147.8  217.91  5167.5  219.97  5217.9  225.34  5342.3  229.58
#Mann= 7 ,-1 , 0
  4030.2     .05       0  4451.8      .1       0  4878.1     .12       0
  4994.6     .07       0  5000.6     .12       0  5052.9      .1       0
  5167.5     .05       0
Bank Sta=4707,5067.7
XS Rating Curve= 0 ,0
Exp/Cntr=0.3,0.1

Type RM Length L Ch R = 1 ,21719   ,348,348,348
BEGIN DESCRIPTION:
UNT027 IN PECR 36.0
END DESCRIPTION:
XS GIS Cut Line= 3
       2286829.2     13197013.41      2286782.33     13196659.27
      2286693.79       13195727.
#Sta/Elev= 30
  4065.5  224.57  4102.4  224.68  4233.5  221.82    4263  219.12  4304.1  218.93
  4334.4  217.21  4341.5  216.11  4478.6  212.15  4522.5  210.33  4565.8  211.36
    4616  211.06  4625.6  210.35  4676.3  209.38  4681.8  209.24    4827  207.13
  4880.6  207.37  4967.6  206.96  4987.7  205.78  4994.7  203.82  4997.5  203.32
  5000.7  203.82  5007.8  205.88  5042.7  209.48  5148.4  215.66  5156.2  216.61
  5161.2  216.24  5189.8  217.73  5299.1  223.77  5356.7  224.87  5359.2  224.87
#Mann= 9 ,-1 , 0
  4065.5     .05       0  4478.6     .12       0  4681.8      .1       0
  4880.6     .12       0  4994.7     .07       0  5000.7     .12       0
  5042.7      .1       0  5189.8     .05       0  5356.7      .1       0
Bank Sta=4676.3,5042.7
XS Rating Curve= 0 ,0
Exp/Cntr=0.3,0.1

Type RM Length L Ch R = 1 ,21371   ,541,541,541
BEGIN DESCRIPTION:
UNT027 IN PECR 35.0
END DESCRIPTION:
XS GIS Cut Line= 3
      2287037.72     13196846.87      2287037.72     13196196.85
      2286837.74      13195646.9
#Sta/Elev= 30
  4359.7  223.75  4439.7  220.41  4499.7  215.04  4559.7  211.62  4619.7  209.64
  4638.7  209.86  4709.7  207.11  4779.4  207.31  4799.7  206.96  4809.7  206.03
  4839.7  203.72  4849.7  204.96  4939.7  206.42  4959.7  204.93  4979.7  204.81
  4996.7  201.42  4999.5  200.92  5002.7  201.42  5007.2  202.47  5019.7  202.68
  5041.6  205.79  5050.3  206.03  5051.9  206.05  5150.9  210.03  5166.2  210.77
  5228.5   213.2  5259.1  213.02  5392.8   217.5  5477.9  218.97  5594.9  222.31
#Mann= 8 ,-1 , 0
  4359.7     .05       0  4638.7     .12       0  4779.4     .16       0
  4996.7     .07       0  5002.7     .16       0  5051.9      .1       0
  5150.9     .12       0  5166.2     .05       0
Bank Sta=4809.7,5050.3
XS Rating Curve= 0 ,0
Exp/Cntr=0.3,0.1

Type RM Length L Ch R = 1 ,20830   ,648,648,648
BEGIN DESCRIPTION:
UNT027 IN PECR 34.0
END DESCRIPTION:
XS GIS Cut Line= 3
       2287442.3     13197031.84      2287317.31       13196393.
      2286963.13     13195642.98
#Sta/Elev= 30
  4471.5  222.18  4624.9  219.06  4836.1  218.88  4853.6  217.65  4882.5  212.02
  4975.9  205.29  4990.6  203.45  4996.3  198.05  5003.4  197.64  5006.2  197.14
  5009.4  197.64  5039.5  202.51    5088  205.83  5156.8  205.94  5225.1  203.29
  5246.1   200.2  5270.6  199.96  5298.9   202.5    5390  204.96  5412.7  206.44
  5418.3  208.42  5435.5  208.42    5441  211.18    5481  210.02  5486.6  207.23
  5496.3  207.61  5583.2     212  5674.3  214.42  5742.6  214.44  5951.9  218.91
#Mann= 6 ,-1 , 0
  4471.5     .05       0  5003.4     .03       0  5009.4     .05       0
  5039.5     .16       0  5246.1      .1       0  5496.3     .05       0
Bank Sta=4975.9,5390
XS Rating Curve= 0 ,0
Exp/Cntr=0.3,0.1

Type RM Length L Ch R = 1 ,20182   ,465,465,465
BEGIN DESCRIPTION:
Mapping XS 5b463697
END DESCRIPTION:
XS GIS Cut Line= 3
      2287921.49     13196570.11      2287567.31     13196052.72
      2286924.95       13195393.
#Sta/Elev= 30
  4526.2  216.98    4820   210.3  4866.5  207.81  4918.7  204.33  4978.4   203.1
  4984.4  201.78  4999.4  195.61  5002.4  195.37  5005.2  194.87  5008.4  195.37
  5014.3  200.68  5020.3  201.11  5063.4  202.04  5157.1  201.43  5178.2  203.87
  5206.5  205.21    5274  203.49  5298.6  203.07  5362.1  204.14  5416.5   205.6
  5496.4  208.72    5546  209.75    5553  210.64  5666.5  213.01  5793.5  216.98
  5833.8  217.51  5930.1  221.07  5975.2  222.21  6012.8  224.15    6074  225.84
#Mann= 10 ,-1 , 0
  4526.2     .05       0  4866.5     .16       0  5002.4     .07       0
  5008.4     .16       0    5274     .05       0  5416.5      .1       0
  5666.5     .05       0  5833.8      .1       0  5930.1     .05       0
  5975.2      .1       0
Bank Sta=4918.7,5362.1
XS Rating Curve= 0 ,0
Exp/Cntr=0.3,0.1

Type RM Length L Ch R = 1 ,19717   ,420,420,420
BEGIN DESCRIPTION:
UNT027 IN PECR 33.0
END DESCRIPTION:
XS GIS Cut Line= 3
      2287928.42     13196358.29      2287796.48     13195837.45
       2287105.5     13195278.41
#Sta/Elev= 30
  4340.6  212.78  4529.3  210.11  4575.4  209.41    4632  209.28  4806.3  209.31
    4897  205.69  4927.8  204.07  4969.5  199.13  4976.8  199.19  4983.9  198.62
  4991.9  194.37  4995.3  193.64    4998  193.14  5001.3  193.64  5004.9  193.77
  5012.7  198.87  5019.1  200.25  5033.5   201.1  5069.2  201.76  5142.8  200.02
  5190.2  201.36  5239.7  200.78  5268.5  202.11  5282.9  204.11  5337.5  209.22
  5403.7  212.91  5485.2  215.78  5603.1  218.95  5760.1  222.63  5766.7  222.79
#Mann= 13 ,-1 , 0
  4340.6     .05       0  4529.3      .1       0  4575.4     .05       0
    4632      .1       0    4897     .12       0  4976.8     .16       0
  4995.3     .07       0  5001.3     .16       0  5142.8      .1       0
  5337.5     .05       0  5485.2      .1       0  5603.1     .05       0
  5760.1      .1       0
Bank Sta=4927.8,5282.9
XS Rating Curve= 0 ,0
Exp/Cntr=0.3,0.1

Type RM Length L Ch R = 1 ,19297   ,281,281,281
BEGIN DESCRIPTION:
UNT027 IN PECR 32.0
END DESCRIPTION:
XS GIS Cut Line= 3
      2288008.28     13196313.13      2287841.62     13195844.39
      2287897.15     13195101.55
#Sta/Elev= 30
    4127   212.8  4250.4     211  4270.8  210.09  4376.8  208.67  4439.7  208.68
  4568.8  208.93  4690.1  206.48  4762.4  203.25  4802.5  202.75  4887.8  199.52
  4922.9  198.57  4932.9  199.19  4952.9  198.26    4983  199.14  4993.1   197.9
  5000.1     195  5002.8   194.5  5006.1     195  5013.1   198.6  5033.2  199.42
  5039.9  202.19  5044.9  201.45  5053.2  201.67  5063.2  203.13  5123.4  207.45
  5159.8  208.78  5253.8  212.89  5314.4  214.74    5344  214.82  5369.4  216.34
#Mann= 9 ,-1 , 0
    4127     .05       0  4270.8      .1       0  4376.8     .05       0
  4439.7      .1       0  4690.1     .12       0  4887.8     .16       0
  5000.1     .07       0  5006.1     .16       0  5159.8      .1       0
Bank Sta=4802.5,5063.2
XS Rating Curve= 0 ,0
Exp/Cntr=0.3,0.1

Type RM Length L Ch R = 1 ,19016   ,232,232,232
BEGIN DESCRIPTION:
Mapping XS c2ba3827
END DESCRIPTION:
XS GIS Cut Line= 2
      2288178.17     13196247.85      2288079.33     13195020.22
#Sta/Elev= 30
  4245.5  211.95  4335.4  210.52  4410.9  209.55  4447.1  208.98  4467.2   209.5
  4497.3  208.19  4527.4  208.17  4690.1  203.89    4718   202.4  4788.2  201.23
  4908.6  199.67  4918.7  200.72  4928.7   200.4  4935.1  198.31  4943.2  198.26
  4988.9  196.88  4995.9  194.31  4998.7  193.81  5001.9  194.31    5009  194.74
    5019  198.03    5029  197.11  5062.6  197.72  5079.2   196.9  5104.6  200.87
  5109.3  201.24  5159.4  203.63  5252.1  211.39  5380.2  218.52  5477.1  221.65
#Mann= 8 ,-1 , 0
  4245.5      .1       0  4335.4     .05       0  4410.9      .1       0
  4943.2     .16       0  4995.9     .07       0  5001.9     .16       0
  5104.6      .1       0  5252.1     .05       0
Bank Sta=4788.2,5109.3
XS Rating Curve= 0 ,0
Exp/Cntr=0.3,0.1

Type RM Length L Ch R = 1 ,18784   ,150,150,150
BEGIN DESCRIPTION:
UNT027 IN PECR 31.0
END DESCRIPTION:
XS GIS Cut Line= 2
      2288397.17     13196271.48      2288315.65     13195085.98
#Sta/Elev= 30
  4168.6  211.76  4223.4  211.29  4230.9  210.74  4253.4  210.97    4379   208.1
    4384  208.94  4423.8  208.64    4522  204.84  4527.1  205.37  4564.2  204.16
  4575.5  203.19  4604.3  202.74  4614.3  201.79  4644.3  201.41  4670.1  200.28
  4675.1  200.63  4704.5  199.87  4813.2   198.6    4915  198.25    4935  196.22
  4975.1  197.23  4985.1  196.62  4992.2  195.21  4994.9  194.71  4998.2  195.21
  5104.3  199.82  5135.5   202.4  5143.1  202.23  5265.8  210.26  5356.9   213.4
#Mann= 5 ,-1 , 0
  4168.6     .05       0  4575.5      .1       0  4992.2     .07       0
  4998.2      .1       0  5143.1     .05       0
Bank Sta=4704.5,5104.3
XS Rating Curve= 0 ,0
Exp/Cntr=0.3,0.1

Type RM Length L Ch R = 1 ,18634   ,300,300,300
BEGIN DESCRIPTION:
Mapping XS cd6aacb3
END DESCRIPTION:
XS GIS Cut Line= 3
      2288495.88     13196237.43      2288464.62     13195075.94
      2288464.62     13194846.75
#Sta/Elev= 30
  4136.3  212.23  4189.6  210.79    4447  207.07    4607  199.82  4737.1  198.05
  4836.1  197.97  4907.2  196.31  4957.2  196.78  5004.2  196.04  5006.9  195.54
  5010.2  196.04  5087.2  197.72  5097.2  199.22  5117.2  201.35  5167.3  203.69
  5177.3  205.57  5227.3  208.15  5237.3   209.8  5277.3  210.95  5295.3   212.7
  5337.3   212.9  5347.3  210.44  5367.3  211.06  5387.3  212.81  5407.3  217.55
  5417.3  218.22  5427.3  220.36  5447.3  220.02    5485  221.43  5527.4   223.7
#Mann= 7 ,-1 , 0
  4136.3     .05       0  4189.6      .1       0  4836.1     .05       0
  5004.2     .04       0  5010.2     .05       0  5367.3      .1       0
    5485     .05       0
Bank Sta=4737.1,5097.2
XS Rating Curve= 0 ,0
Exp/Cntr=0.3,0.1

Type RM Length L Ch R = 1 ,18334   ,814,814,814
BEGIN DESCRIPTION:
UNT027 IN PECR 30.0
END DESCRIPTION:
XS GIS Cut Line= 3
      2288570.78     13196288.83      2288745.58     13195428.29
      2288637.71     13194846.82
#Sta/Elev= 30
  3902.1   212.6  4032.6  210.61  4107.9  209.12  4158.6  206.47  4332.7  200.92
    4513  197.23  4557.2  196.49  4587.8  194.72  4638.8  196.16  4791.9  193.91
  4832.5  193.34  4842.7  194.41  4873.2  195.02  4924.1   195.1  4944.4  194.72
  4954.6  192.04    4960  191.58  4985.1  193.94  5002.4  191.39  5005.2  190.89
  5008.4  191.39  5012.9  200.55  5017.9  200.11  5023.8  202.37  5035.9  203.56
  5147.8  206.99  5168.2  209.04  5234.4  211.55  5269.9  215.07  5371.6  221.19
#Mann= 6 ,-1 , 0
  3902.1     .05       0  4032.6      .1       0  4791.9     .12       0
  5002.4     .07       0  5008.4     .12       0  5023.8      .1       0
Bank Sta=4513,5012.9
XS Rating Curve= 0 ,0
Exp/Cntr=0.3,0.1

Type RM Length L Ch R = 1 ,17520   ,573,573,573
BEGIN DESCRIPTION:
UNT027 IN PECR 29.0
END DESCRIPTION:
XS GIS Cut Line= 3
       2289018.7     13196070.08      2289077.73     13195549.25
      2288997.93      13194661.1
#Sta/Elev= 30
  4658.7  210.32  4682.1  210.28  4811.7   206.3  4853.2  206.11  4943.7  203.07
  4959.8  201.75  4964.9  199.44  4973.9  197.12    4984  189.98  4991.1  188.56
  4993.8  188.06  4997.1  188.56  5014.2  192.43  5024.3   191.4  5084.6  192.59
  5094.7  191.55  5114.8  192.75  5131.6   192.5  5139.2  192.38  5155.1  193.55
  5231.9  194.07  5285.7  195.48  5386.1  195.84  5446.3  197.51  5532.1  198.09
  5737.5  201.54    5868   205.9  5906.2  206.56  5918.2  207.45  6074.6  210.29
#Mann= 7 ,-1 , 0
  4658.7     .05       0  4811.7      .1       0  4991.1     .07       0
  4997.1      .1       0  5131.6     .16       0  5231.9     .12       0
  5532.1      .1       0
Bank Sta=4973.9,5285.7
XS Rating Curve= 0 ,0
Exp/Cntr=0.3,0.1

Type RM Length L Ch R = 1 ,16947   ,1185,1185,1185
BEGIN DESCRIPTION:
UNT027 IN PECR 28.0
END DESCRIPTION:
XS GIS Cut Line= 4
      2289327.73     13196031.89      2289473.56     13195611.75
      2289327.73     13195365.22      2289460.46      13194605.9
#Sta/Elev= 30
  4378.8  211.06  4608.4  204.28  4745.1  198.41  4830.1  193.79  4861.4   192.1
  4867.2  190.41  4984.2  189.17  4996.8  186.04  4999.6  185.54  5002.8  186.04
  5005.6  187.76  5015.1  189.32  5027.1  189.81  5036.9  193.13    5050  193.54
  5189.5  196.99  5230.1  196.54  5250.2     193  5260.6  193.94    5291  194.35
  5309.7  196.23  5314.8  194.18  5341.8  198.27  5428.7  199.75  5504.2  198.41
  5547.7  201.43  5658.5  205.41  5737.7  209.48  5808.8  219.51  5880.8   222.4
#Mann= 6 ,-1 , 0
  4378.8     .05       0  4608.4      .1       0  4745.1     .12       0
  4996.8     .07       0  5002.8     .12       0  5658.5      .1       0
Bank Sta=4830.1,5260.6
XS Rating Curve= 0 ,0
Exp/Cntr=0.3,0.1

Type RM Length L Ch R = 1 ,15762   ,344,344,344
BEGIN DESCRIPTION:
UNT027 IN PECR 27.0
END DESCRIPTION:
XS GIS Cut Line= 4
      2289549.93      13196035.4      2289949.25     13195292.31
      2289945.78     13194938.14      2289834.95     13194661.07
#Sta/Elev= 30
  4087.3  211.55  4118.5  210.24  4189.7  207.67  4343.9  200.75  4578.6  193.65
    4645  191.04    4676  190.51  4705.1  188.59  4770.8  189.66  4836.6  187.71
  4852.8  188.67  4858.5  187.83    4891  190.02  4956.4  190.24  4976.4  187.27
  4993.4  182.51  4996.1  182.01  4999.4  182.51  5006.4  186.14  5036.4  187.11
  5056.4  186.38  5066.4  190.36  5086.4  187.99  5106.4  189.45  5116.4  188.37
  5126.4  188.76  5136.4  191.28  5236.6  193.79  5361.9  198.75  5583.5  211.54
#Mann= 7 ,-1 , 0
  4087.3      .1       0  4118.5     .05       0  4189.7      .1       0
  4578.6     .12       0  4993.4     .07       0  4999.4     .12       0
  5236.6      .1       0
Bank Sta=4645,5136.4
XS Rating Curve= 0 ,0
Exp/Cntr=0.3,0.1
