HEC-RAS study RAMIRENA CREEK.prj: RAMIRENA CREEK Base Level Engineering

--- RAMIRENA CREEK.g01 (geometry) --- (continued)

Type RM Length L Ch R = 1 ,46991   ,970,970,970
BEGIN DESCRIPTION:
RAMIRENA CREEK 39.0
END DESCRIPTION:
XS GIS Cut Line= 3
      2283037.71     13235146.85      2282237.72     13234246.85
      2281837.76     13233946.88
#Sta/Elev= 30
  3823.2  190.92  4262.6   157.1  4375.5  150.58  4460.8  148.65  4609.7   151.8
  4786.5  149.34  4822.1  145.91  4885.6  146.87  4899.8  145.35  4906.9   140.1
    4927  136.07  4949.2  134.22  4956.7  130.48    5003  128.97  5005.8  128.47
    5009  128.97  5049.2   130.4  5055.5  134.42  5063.8  132.84  5084.6  135.61
  5090.9  140.62  5099.2  140.73  5105.5  146.87  5120.1   150.6  5152.7  151.77
  5198.9  154.07  5272.7  157.93  5370.3  161.16  5449.2  164.46  5527.3  164.21
#Mann= 8 ,-1 , 0
  3823.2      .1       0    4927     .05       0    5003    .035       0
    5009     .05       0  5152.7      .1       0  5198.9     .16       0
  5272.7      .1       0  5370.3     .05       0
Bank Sta=4906.9,5090.9
XS Rating Curve= 0 ,0
Exp/Cntr=0.3,0.1

Type RM Length L Ch R = 1 ,46021   ,878,878,878
BEGIN DESCRIPTION:
RAMIRENA CREEK 38.0
END DESCRIPTION:
XS GIS Cut Line= 3
      2283137.73      13234346.9      2283037.72     13233846.85
       2282037.7     13232846.83
#Sta/Elev= 30
  4479.2  170.74  4499.6  172.56    4571  172.31  4693.4  167.12  4713.8   162.3
  4805.6  156.72  4815.8  154.05  4856.6  153.66  4907.6  147.26    4928  141.02
  4938.2  133.83  4958.6   132.1  4968.8  129.08  5000.3  127.38    5003  126.88
  5006.3  127.38  5059.9  131.83  5088.1   142.2  5102.3  147.02  5229.6   143.1
  5257.9  147.26    5371  150.29  5512.4  151.87  5581.8  150.06  5715.7  146.82
  5851.8  148.78  6092.2  156.98  6243.5  166.44  6387.5  174.79  6403.4  176.43
#Mann= 7 ,-1 , 0
  4479.2      .1       0  5000.3     .07       0  5006.3      .1       0
  5581.8     .05       0  5715.7      .1       0  6243.5     .08       0
  6387.5      .1       0
Bank Sta=4928,5088.1
XS Rating Curve= 0 ,0
Exp/Cntr=0.3,0.1

Type RM Length L Ch R = 1 ,45143   ,649,649,649
BEGIN DESCRIPTION:
RAMIRENA CREEK 37.0
END DESCRIPTION:
XS GIS Cut Line= 3
      2283387.72     13233496.85      2283287.72     13232996.85
      2282687.74     13232396.87
#Sta/Elev= 30
  4518.4  161.23  4630.6  156.93  4661.2     157  4742.8  152.38  4752.9  152.97
  4763.1  151.75  4793.7  144.36  4820.2  144.42  4844.7  145.75  4875.3  141.73
  4885.5  136.42  4895.7     134  4916.1  134.15  4924.2  132.09  4956.9  126.35
  4984.5  124.46  4987.3  123.96  4990.5  124.46  5031.8  125.12  5070.7  134.09
  5084.9  134.28    5099  139.73  5127.3  141.99  5282.9  144.62  5367.7   143.8
  5424.3  145.14  5480.8  148.26  5751.7  168.94  5752.8  169.02  5876.8   176.9
#Mann= 7 ,-1 , 0
  4518.4      .1       0  4820.2     .16       0  4924.2      .1       0
  4984.5     .07       0  4990.5      .1       0  5751.7     .05       0
  5752.8      .1       0
Bank Sta=4875.3,5099
XS Rating Curve= 0 ,0
Exp/Cntr=0.3,0.1

Type RM Length L Ch R = 1 ,44494   ,614,614,614
BEGIN DESCRIPTION:
Mapping XS abf543f6
END DESCRIPTION:
XS GIS Cut Line= 4
       2283429.7     13233482.43      2283705.73     13233102.25
      2283992.18     13232972.04       2284367.2     13232716.82
#Sta/Elev= 30
  4349.8  158.97  4553.7  149.69  4639.5  138.78  4710.6  143.94  4775.6  144.22
  4811.1  142.19  4819.6  138.77  4909.7   129.6  4967.8  128.31  4990.9  125.15
  4994.6  122.72  4997.3  122.22  5000.6  122.72  5008.5  122.74    5029  134.86
    5037  140.07  5052.5  146.17  5083.2  147.76  5137.5  157.04  5185.6  170.33
  5191.7  168.59  5200.6  170.14  5206.6  167.67  5221.5  172.82  5227.6  171.87
  5236.5  177.93  5242.5  176.26  5257.5  181.28  5371.3  187.25  5587.9  188.09
#Mann= 5 ,-1 , 0
  4349.8      .1       0  4994.6     .07       0  5000.6      .1       0
    5029     .16       0  5137.5      .1       0
Bank Sta=4819.6,5037
XS Rating Curve= 0 ,0
Exp/Cntr=0.3,0.1

Type RM Length L Ch R = 1 ,43880   ,646,646,646
BEGIN DESCRIPTION:
RAMIRENA CREEK 36.0
END DESCRIPTION:
XS GIS Cut Line= 2
      2283432.13     13233612.17      2284374.38     13233590.51
#Sta/Elev= 30
  4682.1  161.65  4694.2  159.44  4767.7   153.8  4927.8  145.84  4947.8  133.57
  4957.8  126.57  4967.5  126.86  4974.2  126.72  4997.8  126.46  5017.8   128.3
  5027.8  127.66  5034.8  125.58  5037.5  125.08  5040.8  125.58  5057.8  127.58
  5073.1  127.65  5076.5   127.4  5107.8  127.74  5131.9  130.83  5137.8  133.09
  5147.8  136.32  5237.8   143.5  5287.8  159.23  5347.9  164.78  5407.9  168.18
  5437.9   176.1  5507.9  180.54  5517.9  182.87  5564.5  186.78  5624.6  186.94
#Mann= 7 ,-1 , 0
  4682.1      .1       0  4967.5     .16       0  4974.2      .1       0
  5034.8     .07       0  5040.8      .1       0  5073.1     .16       0
  5076.5      .1       0
Bank Sta=4947.8,5137.8
XS Rating Curve= 0 ,0
Exp/Cntr=0.3,0.1

Type RM Length L Ch R = 1 ,43234   ,927,927,927
BEGIN DESCRIPTION:
RAMIRENA CREEK 35.0
END DESCRIPTION:
XS GIS Cut Line= 3
       2283301.9     13234230.66      2284202.52     13234219.81
      2284387.03     13234132.98
#Sta/Elev= 30
  4631.6   172.2  4637.4  170.83  4787.4   155.3  4869.8  147.57  4897.4   147.2
  4957.4  136.78  4967.4  126.55  4989.9  125.51  5004.4  124.47  5007.2  123.97
  5010.4  124.47  5017.4  126.55  5047.5  126.09  5057.5  127.54  5097.5  129.27
  5137.5  129.56  5177.5  125.65  5197.5  125.88  5207.5  132.68  5217.5  136.47
  5227.5  140.35  5277.5  145.36  5347.5  156.01  5377.5  156.97  5487.5  168.24
  5532.3  173.32    5538  175.29  5552.8  177.49  5621.2  181.23  5736.2  184.48
#Mann= 5 ,-1 , 0
  4631.6      .1       0  4869.8     .16       0  4989.9      .1       0
  5004.4     .07       0  5010.4      .1       0
Bank Sta=4957.4,5217.5
XS Rating Curve= 0 ,0
Exp/Cntr=0.3,0.1

Type RM Length L Ch R = 1 ,42307   ,814,814,814
BEGIN DESCRIPTION:
RAMIRENA CREEK 34.0
END DESCRIPTION:
XS GIS Cut Line= 3
      2283187.73     13235196.85      2283787.72     13235096.85
      2284287.75     13235096.85
#Sta/Elev= 30
  4411.9  185.19  4482.9  177.91    4493  175.83  4543.7  169.65  4622.3  161.13
  4655.2  155.61    4715  149.43    4749  144.98  4766.7  141.52  4804.7  138.22
  4870.6  136.87  4888.4   137.8  4919.6  135.02  4926.4     133  4931.5  133.94
  4939.1  128.69  4959.3  123.33  4979.6  124.08    5007  123.12  5009.8  122.62
    5013  123.12  5030.2  123.98  5050.2   131.5  5060.2  137.38  5070.2  136.68
  5080.2   138.1  5100.2  138.46  5170.2  148.82  5330.2  155.25  5520.2  168.11
#Mann= 5 ,-1 , 0
  4411.9      .1       0    4715     .16       0  4919.6      .1       0
    5007     .07       0    5013      .1       0
Bank Sta=4931.5,5060.2
XS Rating Curve= 0 ,0
Exp/Cntr=0.3,0.1

Type RM Length L Ch R = 1 ,41493   ,659,659,659
BEGIN DESCRIPTION:
RAMIRENA CREEK 33.0
END DESCRIPTION:
XS GIS Cut Line= 3
      2283199.87     13235806.16      2283482.03     13235914.69
      2284293.22     13235866.97
#Sta/Elev= 30
  4410.9  188.95  4440.7  183.98  4455.7  183.31  4462.2   181.7    4565  170.28
    4580  169.92  4644.3   162.2  4697.9  157.68  4704.3  156.01  4819.2  145.47
  4839.1  143.79  4879.2  138.15  4949.3  134.72  4959.3  129.95  4979.4  123.62
  4986.9  123.28  4996.4  121.77  4999.1  121.27  5002.4  121.77  5089.5  124.87
  5103.3  128.56  5109.6   134.6  5129.6  136.11  5179.7  135.96  5229.8  141.16
  5299.9  146.26  5470.2  157.39  5490.2  157.74  5520.3   160.6  5525.8  162.04
#Mann= 5 ,-1 , 0
  4410.9      .1       0  4819.2     .16       0  4986.9      .1       0
  4996.4     .07       0  5002.4      .1       0
Bank Sta=4949.3,5109.6
XS Rating Curve= 0 ,0
Exp/Cntr=0.3,0.1

Type RM Length L Ch R = 1 ,40834   ,504,504,504
BEGIN DESCRIPTION:
Mapping XS d566d330
END DESCRIPTION:
XS GIS Cut Line= 3
       2283000.3     13236439.87      2283421.27     13236565.73
      2284219.88     13236504.97
#Sta/Elev= 30
  4082.6  177.12  4158.8     172  4197.1  171.17    4225   169.3  4296.4  167.39
  4382.6  167.47  4406.2  166.35  4709.4  148.68  4759.1  144.76  4849.4  134.53
  4879.5  134.72  4889.5  132.84  4929.6  132.32  4949.7  129.79  4959.7   122.9
  4996.8  120.51  4999.6  120.01  5002.8  120.51  5019.9  121.97  5039.9  122.22
    5050  124.23    5070  131.72    5080  136.44  5090.1  137.12  5110.1  135.71
  5120.2  136.98  5140.2  137.32  5250.5  148.19  5310.7  152.87  5322.9  152.73
#Mann= 3 ,-1 , 0
  4082.6      .1       0  4996.8     .07       0  5002.8      .1       0
Bank Sta=4929.6,5070
XS Rating Curve= 0 ,0
Exp/Cntr=0.3,0.1

Type RM Length L Ch R = 1 ,40330   ,515,515,515
BEGIN DESCRIPTION:
Mapping XS 14f3a109
END DESCRIPTION:
XS GIS Cut Line= 3
      2282857.08     13236934.66      2283451.65      13237047.5
      2284211.23      13237004.1
#Sta/Elev= 30
  3887.8  170.75  4051.3  163.28  4061.5  163.43  4132.7  158.84    4204  156.59
  4214.2  155.48  4336.3   150.4  4358.6   150.3  4427.9  146.93  4566.6  143.68
  4609.2   143.5  4699.4  140.58  4765.9  135.06  4789.5  134.05  4859.6  133.36
  4909.7  131.48  4919.7  127.64  4938.6  122.72  4949.8  121.79  4996.9  120.83
  4999.6  120.33  5002.9  120.83  5011.5  121.48  5019.9  123.66  5029.9  129.16
  5039.9  132.96    5050  134.32    5080  134.67  5170.2  144.42  5253.8  150.88
#Mann= 5 ,-1 , 0
  3887.8      .1       0  4566.6     .16       0  4996.9     .07       0
  5002.9     .16       0  5011.5      .1       0
Bank Sta=4909.7,5039.9
XS Rating Curve= 0 ,0
Exp/Cntr=0.3,0.1

Type RM Length L Ch R = 1 ,39815   ,247,247,247
BEGIN DESCRIPTION:
Mapping XS b35ca7f7
END DESCRIPTION:
XS GIS Cut Line= 3
      2282856.99     13237333.94      2283260.68     13237503.23
      2284123.52     13237507.56
#Sta/Elev= 30
  3903.7  178.37  3951.7  176.52  4045.5  169.62  4052.2  168.35  4057.6  168.65
  4240.6  155.07  4348.5  148.86  4478.5  143.76  4690.4  139.25  4768.5   135.9
  4948.5  132.08  4955.3  130.62  4968.5  128.11  4978.5  127.45  4988.5  124.25
  4995.5  120.63  4998.2  120.13  5001.5  120.63  5058.5  121.06  5068.5  121.95
  5078.5  125.66  5088.5  127.77  5098.5  131.92  5108.5  134.22  5118.5  135.07
  5138.5  139.61  5148.5   143.4  5168.5  147.66  5188.5  149.72  5204.3  149.59
#Mann= 5 ,-1 , 0
  3903.7      .1       0  4690.4     .16       0  4955.3      .1       0
  4995.5     .07       0  5001.5      .1       0
Bank Sta=4948.5,5098.5
XS Rating Curve= 0 ,0
Exp/Cntr=0.3,0.1

Type RM Length L Ch R = 1 ,39568   ,585,585,585
BEGIN DESCRIPTION:
Mapping XS 51995a6a
END DESCRIPTION:
XS GIS Cut Line= 2
      2283030.67      13238245.4      2284103.79     13237649.23
#Sta/Elev= 30
  3984.5  206.69    4114  200.16    4290  184.57  4298.2  179.52  4303.9  181.63
  4312.9  176.89  4319.9   168.4  4325.6  168.93  4341.7  162.29  4359.7  160.73
  4363.1  160.51    4473   148.3  4541.7  143.38  4621.7  139.76  4840.4   135.3
  4878.2  133.44  4899.9  125.17  4904.3  126.68  4921.6  131.46  4965.1  132.36
  4987.8  124.67  4994.1  119.83  4996.9  119.33  5000.1  119.83  5074.1  121.67
  5084.1  122.01  5113.6  129.74  5127.6  130.95  5165.3  139.56  5212.1  146.41
#Mann= 7 ,-1 , 0
  3984.5      .1       0  4359.7     .16       0  4363.1      .1       0
  4904.3     .16       0  4994.1     .07       0  5000.1     .16       0
  5074.1      .1       0
Bank Sta=4965.1,5127.6
XS Rating Curve= 0 ,0
Exp/Cntr=0.3,0.1

Type RM Length L Ch R = 1 ,38983   ,392,392,392
BEGIN DESCRIPTION:
Mapping XS 422b39b9
END DESCRIPTION:
XS GIS Cut Line= 4
      2283742.18     13239065.79      2284075.52     13238399.12
      2284309.89       13238071.      2284153.63     13237643.88
#Sta/Elev= 30
    4007  171.64  4205.5  156.81  4294.9  153.81  4384.3  146.12  4530.6  139.13
  4804.8  136.26  4834.3  134.95  4869.9  135.42  4920.3  131.72  4935.1  128.12
  4941.2  123.69    4956  122.16  4970.7  118.67  4991.6  118.08  4997.2  116.77
  4999.9  116.27  5003.2  116.77  5027.2  122.18  5062.9  124.64  5074.4  125.18
  5148.9  125.95  5170.7  129.26  5176.2  132.34  5191.9  132.36  5201.4   135.4
  5206.7  134.98  5223.9  138.78  5277.1  141.09  5440.3  141.53  5610.4  146.67
#Mann= 5 ,-1 , 0
    4007      .1       0  4530.6     .16       0  4997.2     .07       0
  5003.2     .16       0  5074.4      .1       0
Bank Sta=4941.2,5062.9
XS Rating Curve= 0 ,0
Exp/Cntr=0.3,0.1

Type RM Length L Ch R = 1 ,38591   ,988,988,988
BEGIN DESCRIPTION:
RAMIRENA CREEK 32.0
END DESCRIPTION:
XS GIS Cut Line= 3
      2285037.67     13238246.85      2284537.72     13238146.85
       2284137.7     13237546.82
#Sta/Elev= 30
  4499.5  184.27    4530  185.61  4591.2   185.1  4652.4  182.99  4703.4  178.77
  4723.8  173.48    4734  163.62  4744.2  160.98  4764.6  151.41    4785  146.91
  4830.9  142.95    4887  135.78  4897.2  129.81  4907.4  125.88  4917.6  124.39
  4958.4  122.37  4968.6  120.04  4996.2  117.75  4998.9  117.25  5002.2  117.75
  5104.3  126.84    5110  128.45  5119.1  128.99  5176.1  133.12  5212.2  137.62
  5269.3  137.67  5333.9  139.95  5550.2  141.14  5701.9  148.83  5730.5  148.95
#Mann= 5 ,-1 , 0
  4499.5      .1       0  4996.2     .07       0  5002.2      .1       0
  5104.3     .16       0  5119.1      .1       0
Bank Sta=4897.2,5110
XS Rating Curve= 0 ,0
Exp/Cntr=0.3,0.1

Type RM Length L Ch R = 1 ,37603   ,922,922,922
BEGIN DESCRIPTION:
RAMIRENA CREEK 31.0
END DESCRIPTION:
XS GIS Cut Line= 3
      2285387.71     13237396.85      2284887.72     13237296.85
      2284187.72     13237396.85
#Sta/Elev= 30
  4490.2     180  4571.8  176.18  4622.8  171.35    4633  164.35  4643.2  160.74
  4653.4  155.09  4673.8  151.33  4704.4  148.22  4734.9  143.31  4857.3  128.75
  4867.5  125.65  4877.7  121.86  4887.9  120.44  4918.5   120.1  4994.5  115.03
  4997.3  114.53  5000.5  115.03  5002.6  115.03  5010.2  118.63  5030.4  121.49
  5040.5  125.38  5050.6  127.23  5060.7  129.49  5070.8   130.2  5161.7  134.93
  5394.1  139.46    5485  138.45  5555.7  140.47  5676.9  149.43  5707.2  150.56
#Mann= 3 ,-1 , 0
  4490.2      .1       0  4994.5     .07       0  5000.5      .1       0
Bank Sta=4867.5,5050.6
XS Rating Curve= 0 ,0
Exp/Cntr=0.3,0.1

Type RM Length L Ch R = 1 ,36681   ,891,891,891
BEGIN DESCRIPTION:
RAMIRENA CREEK 30.0
END DESCRIPTION:
XS GIS Cut Line= 3
      2285487.69     13236846.82      2285187.72     13236446.85
      2284487.71     13235946.85
#Sta/Elev= 30
  4479.9  152.31  4751.7  139.59    4758  138.02  4801.7  134.54  4829.9  130.45
  4866.3  127.87  4872.6  124.22  4893.4  120.02    4908  118.49    4999  114.24
  5001.7  113.74    5005  114.24  5016.7  115.54    5029  122.46  5043.8  126.66
  5050.4  128.87  5065.9  129.89    5088  128.48  5138.4  129.69  5151.9  128.36
  5178.8  128.98  5230.6  131.94  5237.9  133.52  5352.2  133.22  5503.4  135.47
  5559.9  138.12    5625  144.17  5660.1  146.21  5756.7  154.97  5840.1  162.59
#Mann= 7 ,-1 , 0
  4479.9      .1       0    4999     .07       0    5005      .1       0
  5050.4     .12       0  5178.8      .1       0  5660.1     .05       0
  5756.7      .1       0
Bank Sta=4866.3,5043.8
XS Rating Curve= 0 ,0
Exp/Cntr=0.3,0.1

Type RM Length L Ch R = 1 ,35790   ,952,952,952
BEGIN DESCRIPTION:
RAMIRENA CREEK 29.0
END DESCRIPTION:
XS GIS Cut Line= 3
      2286037.73     13236046.86      2285537.72     13235646.85
      2284937.72     13235546.85
#Sta/Elev= 30
  4372.4  165.62  4650.1  139.73  4728.6  135.11  4827.8  133.11    4863  126.91
  4871.1  128.98  4884.7  129.74  4898.3  127.17  4912.7  123.34  4920.7  119.26
  4939.7  117.61  4962.3  117.32  4970.3  115.58  4996.1  114.07  4998.9  113.57
  5002.1  114.07  5073.5  118.94  5110.6   125.5  5114.1  126.43    5120  126.24
  5141.8  125.07  5162.3  123.83  5174.9  126.84  5195.2  127.82  5205.3  126.82
  5215.5  129.04  5316.9  128.88  5410.6  136.35  5539.9  149.04    5621  154.61
#Mann= 7 ,-1 , 0
  4372.4      .1       0  4939.7     .16       0  4996.1     .07       0
  5002.1     .16       0  5110.6      .1       0    5120     .16       0
  5141.8      .1       0
Bank Sta=4898.3,5114.1
XS Rating Curve= 0 ,0
Exp/Cntr=0.3,0.1

Type RM Length L Ch R = 1 ,34838   ,763,763,763
BEGIN DESCRIPTION:
RAMIRENA CREEK 28.0
END DESCRIPTION:
XS GIS Cut Line= 3
      2286287.72     13235496.86      2286087.72     13234996.85
      2286087.72     13234396.88
#Sta/Elev= 30
  4478.8  149.01    4565  147.75  4603.3  144.82  4626.4  142.33  4694.2  134.85
  4748.1  130.39  4771.6  126.99  4801.5  125.02  4816.7  125.38  4823.5  126.87
  4846.3  126.94  4865.2  124.22  4870.6  124.44  4888.1  121.71  4894.8  117.83
    4954  116.02  4963.5  114.12  4992.8  112.63  4995.5  112.13  4998.8  112.63
  5002.5  114.63  5037.3  115.21  5057.3  120.38  5067.3   121.4  5077.3  126.27
  5117.3  129.48  5217.3  129.55  5357.3  136.38  5437.3  141.44  5617.3  158.82
#Mann= 7 ,-1 , 0
  4478.8      .1       0  4603.3     .16       0  4626.4      .1       0
  4771.6     .16       0  4801.5      .1       0  4992.8     .07       0
  4998.8      .1       0
Bank Sta=4870.6,5077.3
XS Rating Curve= 0 ,0
Exp/Cntr=0.3,0.1

Type RM Length L Ch R = 1 ,34075   ,669,669,669
BEGIN DESCRIPTION:
RAMIRENA CREEK 27.0
END DESCRIPTION:
XS GIS Cut Line= 4
      2286489.86     13235654.26      2286641.76     13235515.38
      2286962.94     13234933.78      2286893.71      13234630.9
#Sta/Elev= 30
  4407.9  148.04  4454.2  146.11  4595.4  135.96  4650.3  133.94  4716.8  131.44
  4781.7  129.76  4817.3  127.36  4829.1  124.94  4851.9  126.24  4874.8  123.69
  4892.7  119.48  4954.7  113.31  4997.4  110.84  5000.2  110.34  5003.4  110.84
  5034.9  113.06  5045.3  115.89    5051  117.94  5057.5  125.71  5148.4  124.84
  5175.9  127.74  5213.7  135.73  5263.2  143.15  5346.8  147.73  5377.5  151.22
  5429.7  153.32  5434.8  153.17  5461.7   154.2  5499.5  152.41  5588.8   155.1
#Mann= 9 ,-1 , 0
  4407.9      .1       0  4650.3     .16       0  4716.8      .1       0
  4781.7     .16       0  4892.7      .1       0  4997.4     .07       0
  5003.4      .1       0  5429.7     .08       0  5434.8      .1       0
Bank Sta=4874.8,5057.5
XS Rating Curve= 0 ,0
Exp/Cntr=0.3,0.1

Type RM Length L Ch R = 1 ,33406   ,652,652,652
BEGIN DESCRIPTION:
Mapping XS cfc0bc34
END DESCRIPTION:
XS GIS Cut Line= 3
      2286541.93     13235940.73       2286754.6     13235897.33
      2287739.88     13235463.29
#Sta/Elev= 30
  4225.4   148.4  4342.3  142.67  4453.7   135.5  4551.9  132.05  4660.4  129.97
  4732.2  127.53  4778.8  128.13  4802.2  126.86    4836  128.18  4861.1  126.88
  4877.6  122.46  4893.9  116.17  4919.7  115.05  4953.1   113.6  4970.4  110.49
  5002.2  109.98  5004.9  109.48  5008.2  109.98    5023  116.27  5035.9  119.54
  5051.8  120.47  5057.8  122.37  5090.6  123.73  5179.4  132.29  5188.9  131.88
  5210.8  136.14  5309.1  145.43  5371.5   151.1  5462.1  157.15  5519.1  162.71
#Mann= 8 ,-1 , 0
  4225.4     .05       0  4342.3      .1       0  4551.9     .16       0
  4660.4      .1       0    4836     .16       0  4919.7      .1       0
  5002.2     .07       0  5008.2      .1       0
Bank Sta=4877.6,5057.8
XS Rating Curve= 0 ,0
Exp/Cntr=0.3,0.1

Type RM Length L Ch R = 1 ,32754   ,979,979,979
BEGIN DESCRIPTION:
RAMIRENA CREEK 26.0
END DESCRIPTION:
XS GIS Cut Line= 4
      2286521.96     13236465.03      2286839.67     13236345.24
      2287787.59     13236235.87      2287891.78     13236256.71
#Sta/Elev= 30
  4050.7  170.79  4231.5  159.13  4286.5  154.42  4386.5  142.23  4510.6  132.45
  4579.5  129.15  4690.3  127.22  4811.1  122.75  4830.8  123.71  4871.5  124.95
  4881.5  123.12  4891.6  118.21  4901.7  116.61  4942.9  114.48  4962.1  112.22
  4972.1  109.47  4999.3  109.04  5002.1  108.54  5005.3  109.04  5062.7  119.12
  5072.8  119.79  5082.9  123.53  5117.9  127.28  5123.1  130.87  5153.3  135.66
  5163.4  138.67  5223.8   142.2    5254  146.39  5372.5  155.76  5450.7  156.21
#Mann= 5 ,-1 , 0
  4050.7      .1       0  4830.8     .16       0  4942.9      .1       0
  4999.3     .07       0  5005.3      .1       0
Bank Sta=4871.5,5082.9
XS Rating Curve= 0 ,0
Exp/Cntr=0.3,0.1

Type RM Length L Ch R = 1 ,31775   ,713,713,713
BEGIN DESCRIPTION:
RAMIRENA CREEK 25.0
END DESCRIPTION:
XS GIS Cut Line= 4
       2286245.9     13237063.98      2286574.05     13237235.87
      2287725.09     13237188.99      2287881.34     13237053.58
#Sta/Elev= 30
  3914.4  176.02  3932.4  174.87  3961.6  170.32  4081.2  159.97    4131  156.99
  4198.7   149.7  4378.5  135.97  4508.7  128.89  4748.8  125.02  4808.9   125.6
    4909  123.29    4919  121.75  4939.1  118.22  4949.1  113.26  4969.1  113.56
  4989.1  107.12  5006.1  107.04  5008.9  106.54  5012.1  107.04  5029.1  110.39
  5049.1   112.3  5079.2  111.57  5099.2  113.28  5109.2  118.87  5129.2  122.08
  5149.2  121.43  5214.1   129.4  5279.3     138  5447.3  151.45  5643.6  155.72
#Mann= 5 ,-1 , 0
  3914.4      .1       0  4748.8     .16       0  5006.1     .07       0
  5012.1     .16       0  5214.1      .1       0
Bank Sta=4919,5129.2
XS Rating Curve= 0 ,0
Exp/Cntr=0.3,0.1

Type RM Length L Ch R = 1 ,31062   ,944,944,944
BEGIN DESCRIPTION:
RAMIRENA CREEK 24.0
END DESCRIPTION:
XS GIS Cut Line= 3
      2286287.73     13238096.85      2287287.72     13237896.85
      2287687.73     13237596.85
#Sta/Elev= 30
  3989.7  165.43    4044  161.37  4132.5  154.61  4203.8  146.41  4234.4  145.85
  4358.9  134.97  4489.4   126.8  4603.1  124.76  4693.4     122  4805.5  122.01
  4917.7  117.93  4950.3  113.17  4978.9  107.32  4989.1  107.65  4996.3  105.33
    4999  104.83  5002.3  105.33  5012.6   105.7  5016.8   108.4  5061.3  115.12
    5073  119.75  5137.6  121.75  5181.4  128.92  5202.2  129.35  5209.5  133.05
  5259.5  136.21  5287.6  138.56    5438   144.1  5457.4  144.64  5509.5  145.43
#Mann= 11 ,-1 , 0
  3989.7     .16       0    4044      .1       0  4358.9     .16       0
  4603.1      .1       0  4950.3     .16       0  4996.3     .07       0
  5002.3     .16       0  5061.3     .12       0  5259.5      .1       0
    5438     .12       0  5457.4      .1       0
Bank Sta=4917.7,5073
XS Rating Curve= 0 ,0
Exp/Cntr=0.3,0.1

Type RM Length L Ch R = 1 ,30118   ,931,931,931
BEGIN DESCRIPTION:
RAMIRENA CREEK 23.0
END DESCRIPTION:
XS GIS Cut Line= 3
      2287387.72     13238946.85      2287787.72     13238646.85
      2288087.73     13237746.84
#Sta/Elev= 30
  4496.8  152.29  4624.9  143.63  4768.7  138.49  4804.1   134.9  4883.3   122.7
  4924.9  119.21  4939.5  113.48  4986.5  105.46  4989.3  104.96  4992.5  105.46
    5039  108.07  5049.5  111.45    5060  112.23  5081.1  111.17  5091.7  112.75
  5105.9  117.79  5112.7  119.39  5133.8  122.16  5144.4  125.68  5176.6  125.16
  5228.7  121.19  5270.9   123.4  5291.9  121.88  5323.6  122.87  5365.7  125.66
  5429.4   124.7  5433.7  124.65  5555.5  124.92  5618.7   127.2  5945.5  150.11
#Mann= 7 ,-1 , 0
  4496.8      .1       0  4986.5     .07       0  4992.5      .1       0
  5105.9     .16       0  5176.6      .1       0  5429.4     .16       0
  5433.7      .1       0
Bank Sta=4924.9,5112.7
XS Rating Curve= 0 ,0
Exp/Cntr=0.3,0.1

Type RM Length L Ch R = 1 ,29187   ,1054,1054,1054
BEGIN DESCRIPTION:
RAMIRENA CREEK 22.0
END DESCRIPTION:
XS GIS Cut Line= 3
      2288287.73     13239796.82      2288687.72     13238796.85
      2288787.72     13237896.89
#Sta/Elev= 30
  3895.7  165.21  3914.4   163.6  4003.4  153.71  4311.7  130.38  4419.4   126.1
  4605.2  124.37  4649.6  119.53  4681.9  118.28  4703.4  114.11  4735.7  110.97
  4789.6  114.42  4819.7  114.55  4932.1  105.87  4940.4  105.51  4951.2  108.29
  4957.9  107.45  4975.2  109.66  4989.8  105.14  4992.6  104.64  4995.8  105.14
  5012.9  106.02    5023  109.79  5033.1  117.34  5043.1  120.66  5063.3  122.39
  5123.6  120.29  5254.4  122.59  5465.7  121.44  5596.5  129.44  5878.2  152.22
#Mann= 6 ,-1 , 0
  3895.7     .05       0  3914.4      .1       0  4819.7     .16       0
  4932.1      .1       0  4989.8     .07       0  4995.8      .1       0
Bank Sta=4819.7,5033.1
XS Rating Curve= 0 ,0
Exp/Cntr=0.3,0.1

Type RM Length L Ch R = 1 ,28133   ,701,701,701
BEGIN DESCRIPTION:
RAMIRENA CREEK 21.0
END DESCRIPTION:
XS GIS Cut Line= 4
      2288986.38     13240450.64      2289513.99     13239775.68
      2289656.58     13238777.55      2289234.15     13238151.02
#Sta/Elev= 30
  3588.4  145.72  3862.3  143.58  4126.3  129.28  4148.1  129.36  4183.3  125.83
  4282.8  120.79  4387.7  117.82  4484.3  117.46  4621.2  120.69  4720.6  121.43
  4822.7  119.01  4856.7  116.35  4898.5  117.28    4958   111.1  4989.1  101.49
  5019.7  104.12  5029.8  109.82  5039.9  110.89  5068.8  108.76  5144.6  108.84
  5161.1  114.65  5181.3  117.52  5215.3  117.63    5252  115.19  5329.2  119.36
  5422.4  127.67  5655.1  131.64    5877  144.21  6057.2  140.88    6209  140.12
#Mann= 8 ,-1 , 0
  3588.4      .1       0  4387.7     .12       0  4621.2      .1       0
  4720.6     .16       0  4822.7      .1       0    4958     .07       0
  5029.8     .16       0  5329.2      .1       0
Bank Sta=4958,5039.9
XS Rating Curve= 0 ,0
Exp/Cntr=0.3,0.1

Type RM Length L Ch R = 1 ,27432   ,734,734,734
BEGIN DESCRIPTION:
RAMIRENA CREEK 20.0
END DESCRIPTION:
XS GIS Cut Line= 2
      2290184.16     13240502.85      2290293.48     13238154.89
#Sta/Elev= 30
  3862.3  152.89  4098.6  145.59  4442.4  121.28  4448.1  121.06  4571.1   115.4
  4645.6   114.8  4769.3  118.46  4843.1  117.91  4889.4  116.95  4919.4  112.49
  4939.5  112.26  4949.5  111.12  4969.5  101.27  4979.3  100.32  5009.5  101.21
  5039.6  108.34  5079.6  107.69  5099.6  112.17  5109.6  115.33  5149.7  119.66
  5218.1  119.16  5257.7  119.48  5590.2   118.6  5680.3  120.39  5765.4  125.21
  5766.9   125.2  5890.5  132.05  5910.5  134.82  5940.5  135.22  6212.8  154.73
#Mann= 12 ,-1 , 0
  3862.3      .1       0  4442.4     .16       0  4448.1     .12       0
  4571.1      .1       0  4645.6     .12       0  4843.1      .1       0
  4939.5     .07       0  5099.6      .1       0  5218.1     .16       0
  5257.7      .1       0  5765.4     .12       0  5766.9      .1       0
Bank Sta=4939.5,5099.6
XS Rating Curve= 0 ,0
Exp/Cntr=0.3,0.1

Type RM Length L Ch R = 1 ,26698   ,1213,1213,1213
BEGIN DESCRIPTION:
RAMIRENA CREEK 19.0
END DESCRIPTION:
XS GIS Cut Line= 3
      2290569.13     13240450.64      2290916.12     13239804.19
      2291063.46     13238316.56
#Sta/Elev= 30
    3933   153.3  4023.8  150.19  4289.1  132.77    4407  130.28  4652.3   133.1
  4885.1  127.26  4905.2  125.38  4925.3  119.27  4938.5  111.98  4955.4  109.04
  4985.3  101.05  5015.7  102.71  5045.9  108.15  5118.7  107.45  5140.4  107.49
  5156.4  111.86  5166.5  112.63  5235.2  115.26  5323.8  115.19  5422.8  117.81
    5478  118.52  5578.5  114.29  5675.8  116.91  5819.6  127.49  6000.5  143.72
  6030.7   147.2  6049.2   152.1  6054.2  150.84  6111.1  155.55  6161.6   161.9
#Mann= 8 ,-1 , 0
    3933      .1       0  4955.4     .07       0  5045.9      .1       0
  5118.7     .16       0  5235.2      .1       0  5323.8     .16       0
  5422.8     .12       0  5675.8      .1       0
Bank Sta=4955.4,5045.9
XS Rating Curve= 0 ,0
Exp/Cntr=0.3,0.1

Type RM Length L Ch R = 1 ,25485   ,952,952,952
BEGIN DESCRIPTION:
RAMIRENA CREEK 18.0
END DESCRIPTION:
XS GIS Cut Line= 3
      2291139.52      13240612.2      2291819.19     13240037.09
      2292465.61     13238682.46
#Sta/Elev= 30
  3448.3  142.25  3663.8  124.26  3776.4  117.28    3877  114.18  4002.4   115.1
    4023  114.96  4150.2  116.36  4297.1  117.07  4483.7  115.84  4527.2  118.17
  4638.1  117.37  4651.7  113.88  4691.5  116.17    4771  112.28  4833.2  106.34
  4929.5   107.3  4937.2  106.83  4952.2  101.92  4997.3  100.21  5020.3  101.73
    5043  112.19  5048.5  113.87  5059.1  115.21  5116.6  113.73  5172.3  115.36
  5192.2     116  5258.6  119.17  5575.9  143.13    5644  146.12  5839.6  149.17
#Mann= 11 ,-1 , 0
  3448.3      .1       0  3776.4     .12       0  4002.4      .1       0
    4023     .16       0  4150.2      .1       0  4297.1     .16       0
  4483.7      .1       0    4771     .07       0  5048.5      .1       0
  5172.3     .12       0  5192.2      .1       0
Bank Sta=4771,5043
XS Rating Curve= 0 ,0
Exp/Cntr=0.3,0.1

Type RM Length L Ch R = 1 ,24533   ,667,667,667
BEGIN DESCRIPTION:
RAMIRENA CREEK 17.0
END DESCRIPTION:
XS GIS Cut Line= 3
      2291147.28      13240786.8       2291589.6     13240704.89
        2293088.     13239771.45
#Sta/Elev= 30
  3513.4  144.87    3779   124.1  3890.1  116.25  4004.5  113.13  4210.8  115.45
    4519  116.79    4650  115.36  4690.9  112.72    4715  110.59  4844.7  116.07
  4860.1  115.56  4875.4  110.28  4881.3  110.34  4890.8  104.58  4927.1  106.24
  4954.5  103.83  4962.5  100.47  5012.1   97.51  5056.7  104.34  5064.3  108.23
  5079.6  109.61  5085.5  108.89  5092.1  111.92  5115.6  115.19  5137.4     121
  5143.3     125  5164.6  127.92  5464.8  136.98  5488.5  137.49  5728.6  145.07
#Mann= 8 ,-1 , 0
  3513.4      .1       0    3779     .12       0  4210.8      .1       0
  4690.9     .16       0  4890.8     .07       0  5079.6      .1       0
  5464.8     .16       0  5488.5      .1       0
Bank Sta=4881.3,5079.6
XS Rating Curve= 0 ,0
Exp/Cntr=0.3,0.1

Type RM Length L Ch R = 1 ,23866   ,766,766,766
BEGIN DESCRIPTION:
Mapping XS 7238af6f
END DESCRIPTION:
XS GIS Cut Line= 3
      2291605.97     13241540.42      2292122.04     13241057.12
      2293399.91     13240188.82
#Sta/Elev= 30
  3853.1  145.74  3955.8  140.78  4334.3  112.86  4359.3  111.47  4394.5  103.05
  4472.2  106.53  4514.7  101.73  4528.8  102.25  4565.2  110.85  4586.2  111.79
  4730.5   110.7  4834.4  110.22  4933.7  106.74  4953.9  105.78  4960.4  102.34
  5017.1   97.25  5032.3  103.35  5047.2   100.2  5053.3  101.92  5089.2  100.36
  5119.1  103.57  5147.3  102.67    5176     107  5183.6  108.86    5191  112.51
  5241.8  119.06  5334.7  119.33  5798.9  140.16  5918.4  146.47  6105.1  153.33
#Mann= 9 ,-1 , 0
  3853.1      .1       0  4334.3     .12       0  4730.5     .16       0
  4834.4     .12       0  4933.7     .16       0  4953.9     .07       0
  5183.6      .1       0  5798.9     .16       0  5918.4      .1       0
#XS Ineff= 1 ,-1
 4302.39 4586.91  111.82
Permanent Ineff=
       F
Bank Sta=4953.9,5176
XS Rating Curve= 0 ,0
Exp/Cntr=0.3,0.1

Type RM Length L Ch R = 1 ,23100   ,369,369,369
BEGIN DESCRIPTION:
Mapping XS 9fb0bf8a
END DESCRIPTION:
XS GIS Cut Line= 2
      2291834.43      13242116.8      2293396.91     13240887.65
#Sta/Elev= 30
  4055.8  159.62  4314.5  145.39  4478.9  131.26  4549.4  128.13  4707.8  113.58
  4741.9  109.38  4770.8  108.39  4955.2  107.76  4969.6  104.66  4984.1   99.04
  5004.6   97.13  5033.8  100.13  5083.5  100.66  5097.9     104  5141.3  106.49
  5268.7  109.34  5325.7  111.77  5360.9  114.89  5409.4  113.97  5433.2  112.91
  5560.3  113.38    5568  113.67  5648.9  117.32  5752.2  124.33  5781.1  127.03
    5810  131.53  5938.3  143.57  5959.1  144.02  6002.5  150.01  6043.8  152.67
#Mann= 8 ,-1 , 0
  4055.8      .1       0  4707.8     .12       0  4955.2     .07       0
  5141.3      .1       0  5409.4     .16       0  5560.3      .1       0
    5568     .16       0  5648.9      .1       0
Bank Sta=4955.2,5141.3
XS Rating Curve= 0 ,0
Exp/Cntr=0.3,0.1

Type RM Length L Ch R = 1 ,22731   ,1042,1042,1042
BEGIN DESCRIPTION:
Mapping XS de6fdc89
END DESCRIPTION:
XS GIS Cut Line= 2
       2292240.7     13242325.12      2293511.54     13241106.36
#Sta/Elev= 30
  4328.5  135.02  4417.2  132.95  4438.2  133.82  4473.8  131.55  4622.2   132.3
  4650.5  131.06  4841.4  111.64  4912.2  107.22  4954.6  108.16  4961.7  106.89
  4982.9   98.78  4996.8   97.76  5088.9  101.82  5131.4  105.55  5138.6  106.22
  5329.5  112.84  5395.9  112.92  5407.4  113.04  5506.2  113.79  5543.8  112.76
  5598.4  111.04  5661.9  111.63  5775.1  119.12    5816  123.96  5874.2   129.3
  5881.1   131.1  5937.7  137.03  5959.1  138.17  6001.2  144.28  6089.3  153.98
#Mann= 7 ,-1 , 0
  4328.5      .1       0  4954.6     .07       0  5131.4      .1       0
  5395.9     .16       0  5407.4      .1       0  5543.8     .16       0
    5816      .1       0
Bank Sta=4954.6,5138.6
XS Rating Curve= 0 ,0
Exp/Cntr=0.3,0.1

Type RM Length L Ch R = 1 ,21689   ,1135,1135,1135
BEGIN DESCRIPTION:
RAMIRENA CREEK 14.0
END DESCRIPTION:
XS GIS Cut Line= 3
      2293252.46     13242736.36      2293490.01     13242547.96
      2293866.81     13241245.56
#Sta/Elev= 30
  4383.6  132.87  4571.6  134.14  4650.1  133.22    4679  130.73  4733.7  130.15
  4806.1  122.45  4812.9  116.85  4864.9  114.78  4873.3  111.25  4878.5  111.82
  4885.7  109.63  4912.1  106.26  4917.3  107.05  4945.7  101.02    5000   94.83
  5031.5     100  5083.5    98.6  5095.7  100.57  5114.8  106.13  5124.1  109.13
  5135.6  109.53  5196.6  108.01  5208.4  105.74  5229.3  105.07  5271.1  107.37
  5465.6  110.62  5697.7  127.59  5775.9  136.05  5926.7  149.44  6042.6  157.54
#Mann= 5 ,-1 , 0
  4383.6      .1       0  4917.3     .07       0  5114.8      .1       0
  5271.1     .05       0  5465.6      .1       0
Bank Sta=4917.3,5114.8
XS Rating Curve= 0 ,0
Exp/Cntr=0.3,0.1

Type RM Length L Ch R = 1 ,20554   ,905,905,905
BEGIN DESCRIPTION:
RAMIRENA CREEK 13.0
END DESCRIPTION:
XS GIS Cut Line= 3
      2294202.65      13243195.1      2294497.56     13242818.28
      2294915.32     13241753.39
#Sta/Elev= 30
  4133.7  163.06  4156.9  155.84  4179.2  151.62  4235.3  146.28  4392.6  136.83
  4535.5  129.65  4541.8  130.61  4549.9  128.91  4766.4  115.81  4820.6  111.23
    4845  107.01  4914.5  103.17  4923.7  100.46  4946.7  100.03  4953.5   97.74
  5000.2   96.25  5032.2    98.6  5075.6    97.6  5091.8  100.43  5097.2   99.71
  5107.9  104.26  5140.1  106.66  5183.1  102.94  5301.2  101.11  5322.7  103.34
  5344.2  109.85  5392.8  115.23  5579.9  127.78  5668.6  131.72  5756.1  134.25
#Mann= 4 ,-1 , 0
  4133.7      .1       0  4914.5     .07       0  5097.2     .05       0
  5668.6      .1       0
Bank Sta=4914.5,5107.9
XS Rating Curve= 0 ,0
Exp/Cntr=0.3,0.1

Type RM Length L Ch R = 1 ,19649   ,963,963,963
BEGIN DESCRIPTION:
RAMIRENA CREEK 12.0
END DESCRIPTION:
XS GIS Cut Line= 2
      2295538.11     13243290.34      2295438.93     13241816.88
#Sta/Elev= 30
  4148.1  153.73    4332  137.47  4377.2  132.22  4392.1  131.76  4512.4  121.33
    4763  105.76    4793  105.02    4821   102.2  4843.2  103.49  4863.2  102.29
  4903.3   97.52  5003.3   94.85  5063.7  100.51  5093.7  101.21  5133.8   99.33
  5173.9  103.57    5204  107.25    5234  109.21  5269.9  115.52  5274.9  114.48
  5294.2  117.21  5344.3  120.75  5364.3  123.85  5374.4  123.17  5394.4  126.46
  5419.5  128.41  5497.8  132.02  5534.7  133.76  5594.7  134.17  5624.9   134.3
#Mann= 5 ,-1 , 0
  4148.1      .1       0  4863.2     .07       0  5173.9      .1       0
  5497.8     .08       0  5594.7      .1       0
Bank Sta=4863.2,5173.9
XS Rating Curve= 0 ,0
Exp/Cntr=0.3,0.1

Type RM Length L Ch R = 1 ,18686   ,856,856,856
BEGIN DESCRIPTION:
RAMIRENA CREEK 11.0
END DESCRIPTION:
XS GIS Cut Line= 3
      2296518.35     13243268.46      2296518.35     13242742.46
       2296179.8     13241627.84
#Sta/Elev= 30
  4085.2  138.93  4087.3  138.93  4186.1  135.75  4286.8  130.92  4596.8  109.32
  4697.4  105.53  4773.8  106.12  4787.9   104.8  4826.1  105.66  4892.1  102.74
  4930.6  100.74  4970.9   94.01    5014   91.07  5041.9   94.39  5087.4   94.37
  5107.7  102.62  5118.7  106.14  5129.2  106.63  5160.5  106.25  5178.6  103.01
  5211.5  103.49  5244.1  101.26  5320.6   105.3    5413  107.51  5517.2  113.88
  5561.2  117.24  5588.9  117.11  5670.6  123.12  5720.5  125.33  5776.1  129.21
#Mann= 11 ,-1 , 0
  4085.2      .1       0  4087.3     .05       0  4186.1      .1       0
  4787.9     .16       0  4892.1      .1       0  4930.6     .07       0
  5107.7      .1       0    5413     .05       0  5517.2      .1       0
  5670.6     .08       0  5720.5      .1       0
Bank Sta=4930.6,5107.7
XS Rating Curve= 0 ,0
Exp/Cntr=0.3,0.1

Type RM Length L Ch R = 1 ,17830   ,654,654,654
BEGIN DESCRIPTION:
RAMIRENA CREEK 10.0
END DESCRIPTION:
XS GIS Cut Line= 3
      2297700.42     13243072.23      2297356.37     13242523.39
      2296905.86     13241343.86
#Sta/Elev= 30
  3840.8  158.94  3911.9  154.88    3918  153.58  4237.2  131.37  4664.2  106.44
  4763.2  102.56  4833.9   99.22  4966.6    95.7  5003.4   90.28  5028.4    94.2
  5033.7   97.06  5073.6   96.68    5095   99.38  5113.2    97.3  5127.1   97.02
  5143.3    98.8  5148.6   97.54  5159.2  100.17  5191.4  102.42  5258.2   107.9
    5277  110.88    5313  113.47  5337.7  117.23  5343.1  116.45  5367.8   117.6
  5469.7  124.18  5562.2  127.87  5694.5  130.58  5715.9  132.44  5751.2  131.47
#Mann= 3 , 0 , 0
  3840.8      .1       0  4763.2     .07       0  5191.4      .1       0
Bank Sta=4763.2,5191.4
XS Rating Curve= 0 ,0
Exp/Cntr=0.3,0.1

Type RM Length L Ch R = 1 ,17176   ,1257,1257,1257
BEGIN DESCRIPTION:
RAMIRENA CREEK 9.0
END DESCRIPTION:
XS GIS Cut Line= 3
      2298396.68     13242859.22      2298298.38     13242359.56
      2297013.53     13241001.05
#Sta/Elev= 30
  3657.5  141.09  3863.7  131.03  4006.4  122.95  4036.3  119.69  4047.2  120.91
  4165.6  114.17  4313.7  109.82  4405.7  106.48  4486.4  103.01    4643  101.62
    4721   98.78  4747.4  100.89  4756.3  100.77  4763.1  100.12  4926.2   93.81
  4975.5   95.66  5003.6    92.2  5010.7   95.45  5032.2   98.13  5088.8   100.7
  5095.7  101.03  5173.7  106.09  5208.9  104.02  5314.9  103.93  5428.2  107.67
    5478  107.58  5760.7  118.97  5767.6  120.49  5810.1  120.12  6036.6  132.14
#Mann= 7 ,-1 , 0
  3657.5      .1       0  4313.7     .12       0  4405.7      .1       0
  4486.4     .12       0  4747.4      .1       0  4763.1     .07       0
  5088.8      .1       0
Bank Sta=4756.3,5095.7
XS Rating Curve= 0 ,0
Exp/Cntr=0.3,0.1

Type RM Length L Ch R = 1 ,15919   ,1099,1099,1099
BEGIN DESCRIPTION:
RAMIRENA CREEK 8.0
END DESCRIPTION:
XS GIS Cut Line= 3
      2298871.78     13242023.75      2298871.78     13241499.46
      2298413.21     13239231.14
#Sta/Elev= 30
  4176.7   114.7  4306.1   113.7    4352  113.91    4431  115.06  4637.3  114.64
  4734.3  115.81  4775.1  113.43  4832.3  106.16  4856.7  100.95  4928.1    97.2
  4951.1   96.17  4989.1   91.14  5030.1   94.06  5132.1   96.71  5204.8   95.73
    5275   97.27    5357  103.61  5417.8  102.76  5461.4   99.54  5570.8   93.47
  5723.9   97.98    5975  100.49  6128.4  101.75  6193.2  101.98  6295.2  106.76
  6448.2  116.19  6631.9  129.97  6767.5  131.27  6907.3  136.24  7015.2  138.05
#Mann= 11 ,-1 , 0
  4176.7     .16       0  4306.1      .1       0    4352     .16       0
    4431      .1       0  4637.3     .16       0  4832.3      .1       0
  4928.1     .07       0  5132.1      .1       0  5461.4     .12       0
    5975     .05       0  6128.4      .1       0
Bank Sta=4928.1,5132.1
XS Rating Curve= 0 ,0
Exp/Cntr=0.3,0.1

Type RM Length L Ch R = 1 ,14820   ,372,372,372
BEGIN DESCRIPTION:
RAMIRENA CREEK 7.0
END DESCRIPTION:
XS GIS Cut Line= 3
      2299002.85     13242162.93      2299207.63     13241352.01
      2299379.65     13239631.87
#Sta/Elev= 30
  3075.1  118.92  3118.3  117.82  3436.8  109.72    3615   112.3  3657.5  113.61
  3809.1  116.05  3946.8  110.62  4087.5   98.98  4157.9   97.61  4238.3  101.63
  4258.4   99.77  4263.7   96.85  4298.6   94.31  4426.2   95.56  4464.7   92.63
  4676.9   97.72  4831.2  100.92  4891.5   98.49  4931.7   95.97  4951.5   91.58
  5062.3   92.14  5067.7   97.99  5072.8  101.14  5092.5     104  5112.6  114.74
  5173.3  123.22  5182.9   126.4  5273.8  135.26  5474.8  149.22  5640.2  154.71
#Mann= 10 ,-1 , 0
  3075.1      .1       0  3118.3     .16       0  3436.8      .1       0
    3615     .16       0  3657.5      .1       0  4426.2     .05       0
  4676.9     .12       0  4891.5     .07       0  5072.8      .1       0
  5640.2      .1       0
Bank Sta=4891.5,5067.7
XS Rating Curve= 0 ,0
Exp/Cntr=0.3,0.1

Type RM Length L Ch R = 1 ,14448   ,667,667,667
BEGIN DESCRIPTION:
RAMIRENA CREEK 6.0
END DESCRIPTION:
XS GIS Cut Line= 3
        2299994.     13241966.33      2299682.74     13241089.88
      2299592.71     13239682.13
#Sta/Elev= 30
  3391.4  128.25  3756.5  101.38  3787.2   99.62    3899   96.94  4015.7   97.09
    4154   97.42  4231.9   96.75  4354.6  100.96  4444.8    98.6  4514.9   99.61
  4524.9   99.58    4545   97.02  4625.1   94.19  4675.2   96.99  4775.4   94.05
  4949.6   95.46  5005.6   91.43  5025.9   95.07    5066   96.15  5096.1   99.49
  5108.1  102.04  5116.1  109.52  5126.1  113.38    5165  121.15  5196.3  124.13
  5286.5  127.08  5389.6  135.27  5411.4  136.59    5537  146.34  5732.1  156.28
#Mann= 10 ,-1 , 0
  3391.4      .1       0  3756.5     .12       0  3787.2      .1       0
  4015.7     .12       0    4154      .1       0  4514.9     .07       0
  5096.1     .12       0    5165      .1       0  5389.6     .05       0
  5411.4      .1       0
Bank Sta=4524.9,5096.1
XS Rating Curve= 0 ,0
Exp/Cntr=0.3,0.1

Type RM Length L Ch R = 1 ,13781   ,965,965,965
BEGIN DESCRIPTION:
Mapping XS 521ec740
END DESCRIPTION:
XS GIS Cut Line= 3
      2300291.49     13241315.61      2300280.64     13240621.15
      2300324.05     13239622.83
#Sta/Elev= 30
  4242.9  129.31  4301.7  129.37  4331.7  128.01  4351.7  125.65  4361.7  123.28
  4411.7  118.37  4461.7   111.8  4511.7  107.16  4551.7  102.18  4601.7   98.34
  4661.7   94.11  4711.7   96.16  4721.7   95.17  4771.7   96.11  4841.7   93.73
  4971.8   93.92    4981   92.38  5021.8   93.08  5041.6   91.59  5051.8   93.88
  5071.9   95.29    5172   98.47    5202  100.47  5242.8  101.58  5341.6  104.14
  5462.2  108.01  5736.6  121.35  5752.5  122.04  5762.5  121.12  5936.7     131
#Mann= 6 ,-1 , 0
  4242.9      .1       0  4601.7     .07       0    5172     .12       0
  5242.8     .05       0  5341.6     .12       0  5736.6     .16       0
Bank Sta=4601.7,5172
XS Rating Curve= 0 ,0
Exp/Cntr=0.3,0.1

Type RM Length L Ch R = 1 ,12816   ,610,610,610
BEGIN DESCRIPTION:
RAMIRENA CREEK 5.0
END DESCRIPTION:
XS GIS Cut Line= 4
      2300052.23     13243104.66      2300920.95     13241584.01
      2301190.57     13240539.22      2301050.33     13240051.19
#Sta/Elev= 30
  2663.5  145.83  2960.4   134.1    3230  114.89  3310.6  112.96  3509.3  114.77
  3668.3  108.89  3927.8   96.04    4036   93.35  4172.9    91.6  4175.7    91.1
  4178.9    91.6  4396.2   92.82  4510.5    96.9    4763   96.88  4876.6   92.07
  5072.8   94.29  5100.4   91.89  5176.1   91.99  5269.9   95.27  5298.6    97.9
  5339.3  105.26  5351.7  112.82    5393  128.48  5621.3  140.29  5682.9  140.78
  5725.2  140.74  5860.4  149.39  5952.8  158.73  5964.5  162.38  6001.6  166.67
#Mann= 11 ,-1 , 0
  2663.5      .1       0  3668.3     .16       0  3927.8      .1       0
    4036     .12       0  4172.9     .07       0  4178.9     .12       0
  4510.5      .1       0    4763     .05       0  5269.9      .1       0
  5621.3     .16       0  5682.9      .1       0
Bank Sta=4763,5298.6
XS Rating Curve= 0 ,0
Exp/Cntr=0.3,0.1

Type RM Length L Ch R = 1 ,12206   ,564,564,564
BEGIN DESCRIPTION:
RAMIRENA CREEK 4.0
END DESCRIPTION:
XS GIS Cut Line= 4
      2301024.47     13243773.01      2301583.77     13241567.16
      2301645.56     13240572.93      2301505.13     13240146.03
#Sta/Elev= 30
  2120.7  134.06  2312.3  121.62  2533.6   114.6  2580.8  113.02  2993.6  100.18
  3208.6  106.17  3447.5  103.07    3477  102.05  3681.3   94.54  3846.9   90.74
  3849.6   90.24  3852.9   90.74  4265.1   95.01  4627.1   95.68    4697   92.14
  4997.8   91.96  5138.1   95.75  5204.4   96.03  5392.5  103.53  5483.6  111.12
  5588.4  119.74  5651.1  129.45  5714.7  137.87  5720.8  144.37  5726.1  142.35
  5746.3  154.17  5757.8   155.7  5767.3   162.9  5784.4  169.26  5841.9  172.17
#Mann= 14 ,-1 , 0
  2120.7      .1       0  2533.6     .16       0  2580.8      .1       0
  3447.5     .12       0    3477      .1       0  3681.3     .12       0
  3846.9     .07       0  3852.9     .12       0  4265.1      .1       0
  4627.1     .05       0  5138.1     .12       0  5204.4     .16       0
  5483.6     .05       0  5651.1      .1       0
Bank Sta=4627.1,5138.1
XS Rating Curve= 0 ,0
Exp/Cntr=0.3,0.1

Type RM Length L Ch R = 1 ,11642   ,634,634,634
BEGIN DESCRIPTION:
Mapping XS 94a14cb2
END DESCRIPTION:
XS GIS Cut Line= 3
      2302780.26     13242263.72      2302218.51     13241746.91
      2302111.78     13239926.95
#Sta/Elev= 30
  3484.1  135.44  3554.7  135.34  3674.9  131.78    3866  122.67  3986.3  115.87
  4205.8    98.1  4212.5   97.16  4277.5   92.41  4477.9   92.53  4507.7   90.71
  4588.1   92.68  4808.4   93.93  4998.8    91.8  5169.1   96.16  5202.3   94.63
  5229.2   96.86  5249.2      98  5289.3   91.89  5367.8   93.47  5372.8   92.06
  5427.6   99.99  5499.6  106.53  5538.4  113.75  5569.7  116.47  5790.1  123.26
  5923.3  130.88  6022.4  137.73    6050   140.7    6055  139.84  6070.5  143.17
#Mann= 6 ,-1 , 0
  3484.1      .1       0  4205.8     .05       0  5229.2     .16       0
  5427.6      .1       0  5923.3     .05       0  6022.4      .1       0
Bank Sta=4212.5,5229.2
XS Rating Curve= 0 ,0
Exp/Cntr=0.3,0.1

Type RM Length L Ch R = 1 ,11008   ,672,672,672
BEGIN DESCRIPTION:
RAMIRENA CREEK 3.0
END DESCRIPTION:
XS GIS Cut Line= 3
      2303089.18      13241707.6      2302875.72     13241460.44
       2302342.4     13239877.34
#Sta/Elev= 30
    4279  129.64  4365.6   128.9  4549.9  129.94  4630.5  126.94  4651.6  125.39
  4662.1   122.7  4683.2  120.07    4704  118.95  4714.9  115.14  4740.8  112.15
  4757.1  108.75  4772.3  103.33  4788.7  102.63  4798.5    99.8    4830   98.01
  4835.2   96.51  4841.5   95.23  4861.4   91.99  4883.5   90.71    5137   91.21
  5176.3      93  5221.4    92.1  5307.6   95.18  5496.5   93.27  5611.8   96.39
  5682.8  100.09  5800.9  108.28  6052.8  129.68  6233.1  137.68  6276.1  139.62
#Mann= 5 ,-1 , 0
    4279      .1       0  4841.5     .05       0  5611.8     .12       0
  5682.8      .1       0  6233.1     .05       0
Bank Sta=4835.2,5611.8
XS Rating Curve= 0 ,0
Exp/Cntr=0.3,0.1

Type RM Length L Ch R = 1 ,10336   ,477,477,477
BEGIN DESCRIPTION:
RAMIRENA CREEK 2.0
END DESCRIPTION:
XS GIS Cut Line= 4
      2303268.93      13241623.3      2303437.43     13241011.06
       2302999.3     13240123.55      2302321.39     13239742.58
#Sta/Elev= 30
  4020.4  125.44  4255.3  121.72  4334.6   117.8  4379.7   113.4  4504.2  107.72
  4601.3  106.01  4716.3  107.18  4749.3  106.01  4775.3  102.66  4845.4   94.51
  4887.3   91.21  4890.1   90.71  5182.2   91.21    5240   93.41  5306.9   91.21
  5396.1   91.21  5479.5   94.94  5547.8    98.1  5672.4  103.06  5871.9  115.11
  5893.6  114.68  5974.6  119.49  6128.8  123.96  6264.6  132.53  6325.9  135.56
  6369.7  139.86  6390.9   145.3  6401.1  147.03  6406.8  150.48  6422.8  151.44
#Mann= 7 ,-1 , 0
  4020.4      .1       0  4775.3     .12       0  4887.3     .05       0
  5479.5     .12       0  5547.8      .1       0  6264.6     .05       0
  6390.9      .1       0
Bank Sta=4845.4,5479.5
XS Rating Curve= 0 ,0
Exp/Cntr=0.3,0.1

Type RM Length L Ch R = 1 ,9859    ,181,181,181
BEGIN DESCRIPTION:
Mapping XS 1144e551
END DESCRIPTION:
XS GIS Cut Line= 4
      2303769.27     13241871.16      2303746.45     13240655.86
      2303620.93     13240302.12      2303222.54      13239602.1
#Sta/Elev= 30
  3516.4  123.06  3600.7  122.12  3650.7  120.32  3980.8  100.89  4120.8   95.35
  4178.6    94.1  4240.8   92.19  4376.3   91.86  4475.1   91.96  4540.9   91.82
    4574   92.87  4620.9   94.22  4650.9   92.37  4672.9   92.24  4680.9   92.17
  4697.9   91.21  4700.7   90.71  4703.9   91.21  5251.4   91.21  5288.6    92.9
  5297.4   93.34  5369.3   95.74    5378   97.37    5401   96.68  5427.9    97.8
  5619.6  107.59  5735.4  112.39  5751.2  111.37    5832  110.55  5912.7  110.68
#Mann= 10 ,-1 , 0
  3516.4      .1       0  4178.6     .16       0  4376.3     .12       0
  4475.1     .16       0    4574     .12       0  4672.9     .05       0
  4697.9     .07       0  4703.9     .05       0  5297.4     .16       0
  5427.9      .1       0
Bank Sta=4680.9,5288.6
XS Rating Curve= 0 ,0
Exp/Cntr=0.3,0.1

Type RM Length L Ch R = 1 ,9678    ,226,226,226
BEGIN DESCRIPTION:
Mapping XS 31b6192d
END DESCRIPTION:
XS GIS Cut Line= 3
      2303881.19     13241876.06      2303791.32     13239365.24
      2303712.77     13238501.23
#Sta/Elev= 30
  3469.1  127.71  3548.4  124.49  3709.6  114.53  3878.6  105.59  4034.5   99.03
  4133.5   94.14  4158.7   93.92  4188.8   92.06  4232.4   91.84  4430.4   93.06
    4529   95.14  4544.2   93.67  4628.3    92.4  4669.1   92.26  4679.1   91.92
  4698.8   90.71  5729.7   91.21  5819.8   92.37  5829.8    92.7  6020.1   95.12
  6331.3  103.26  6542.2   106.7  6592.4  108.39  6628.1  111.44  6662.7  112.87
  6672.7  114.61    6723  116.83  6753.1  119.87  6813.3  121.53  6849.1  124.12
#Mann= 9 ,-1 , 0
  3469.1      .1       0  4034.5     .16       0  4133.5      .1       0
  4232.4     .16       0  4430.4     .08       0  4628.3     .05       0
  4669.1     .07       0  4679.1     .05       0  5829.8      .1       0
Bank Sta=4669.1,5819.8
XS Rating Curve= 0 ,0
Exp/Cntr=0.3,0.1

Type RM Length L Ch R = 1 ,9452    ,338,338,338
BEGIN DESCRIPTION:
Mapping XS b1b29180
END DESCRIPTION:
XS GIS Cut Line= 4
      2304100.18     13241819.75      2304043.13     13240148.08
      2304242.82     13239771.52      2304396.91     13239720.15
#Sta/Elev= 30
  3501.7   123.4  3654.7  118.04  3684.7  113.93  3725.1  113.54  3804.8   107.8
  3934.8  100.22  4004.9   97.99  4011.8   96.71  4016.8   97.52    4125   92.27
    4155   92.09    4172   91.21  4174.7   90.71    5187   91.21  5193.8   92.17
  5237.7   91.98  5266.3   94.02  5303.7   94.82    5364   99.05  5402.1   100.5
    5408  101.91  5424.3  101.81  5439.4  103.67    5452  103.56  5458.7  105.09
    5504  108.57  5583.9  113.55  5637.4  116.33  5694.9  117.26    5763  120.74
#Mann= 4 ,-1 , 0
  3501.7     .08       0    4172    .033       0  5193.8     .12       0
  5439.4      .1       0
Bank Sta=4155,5193.8
XS Rating Curve= 0 ,0
Exp/Cntr=0.3,0.1
