--- SALT BRANCH RAMIRENA CREEK.prj (project) ---

Proj Title=SALT BRANCH RAMIRENA CREEK Base Level Engineering
Current Plan=p01
Default Exp/Contr=0.3,0.1
English Units
Geom File=g01
Flow File=f01
Plan File=p01
Y Axis Title=Elevation
X Axis Title(PF)=Main Channel Distance
X Axis Title(XS)=Station
BEGIN DESCRIPTION:
SALT BRANCH RAMIRENA CREEK
END DESCRIPTION:
DSS Export Rating Curves= 0
DSS Export Rating Curve Sorted= 0
DSS Export Volume Flow Curves= 0
DXF OffsetX= 0
DXF OffsetY= 0
DXF ScaleX= 1
DXF ScaleY= 10

--- SALT BRANCH RAMIRENA CREEK.p01 (plan) ---

Plan Title=Multiple Run
Program Version=4.10
Short Identifier=Multiple
Geom File=g01
Flow File=f01
Subcritical Flow
K Sum by GR= 0
Std Step Tol= 0.01
Critical Tol= 0.01
Num of Std Step Trials= 20
Max Error Tol= 0.3
Flow Tol Ratio= 0.001
Split Flow NTrial= 30
Split Flow Tol= 0.02
Split Flow Ratio= 0.02
Log Output Level= 0
Friction Slope Method= 1
Unsteady Friction Slope Method= 2
Unsteady Bridges Friction Slope Method= 1
Parabolic Critical Depth
Global Vel Dist= 1 , 1 , 1
Global Log Level= 0
CheckData=True
Encroach Param=-1 ,0,0, 0
BEGIN DESCRIPTION:
Multiple Run
END DESCRIPTION:
Computation Interval=1HOUR
Output Interval=1HOUR
Run HTab= 0
Run UNet= 0
Run PostProcess= 0
Run WQNet= 0
UNET Theta= 1
UNET Theta Warmup= 1
UNET ZTol= 0.02
UNET ZSATol= 0.05
UNET MxIter= 20
UNET MaxInSteps= 0
UNET DtIC= 0
UNET DtMin= 0
UNET MaxCRTS= 20
UNET WFStab= 2
UNET SFStab= 1
UNET WFX= 1
UNET SFX= 1
UNET DSS MLevel= 4
UNET DZMax Abort= 100
UNET Convert EG Bridges= 0
UNET Use Existing IB Tables=-1
UNET Froude Reduction=False
UNET Froude Limit= 1
UNET Froude Power= 10
UNET Time Slicing=0,0, 5
UNET Junction Losses=0
Instantaneous Interval=1HOUR
Write IC File= 0
Write IC File at Sim End=0
Echo Input=False
Echo Parameters=False
Echo Output=False
Write Detailed= 0
WQ AD Non Conservative
WQ ULTIMATE=-1
WQ Max Comp Step=1HOUR
WQ Output Interval=15MIN
WQ Output Selected Increments= 0
WQ Output face flow=0
WQ Output face velocity=0
WQ Output face area=0
WQ Output face dispersion=0
WQ Output cell volume=0
WQ Output cell surface area=0
WQ Output cell continuity=0
WQ Output cumulative cell continuity=0
WQ Output face conc=0
WQ Output face dconc_dx=0
WQ Output face courant=0
WQ Output face peclet=0
WQ Output face adv mass=0
WQ Output face disp mass=0
WQ Output cell mass=0
WQ Output cell source sink temp=0
WQ Output cell source sink nsm=0
WQ Output MaxMinRange=-1
WQ Daily Max Min Mean=-1
WQ Daily Range=0
WQ Daily Time=0
WQ Create Restart=0
WQ Fixed Restart=0
WQ System Summary=0
WQ Use Fixed Temperature=0
Sorting and Armoring Iterations= 10
XS Update Threshold= 0.02
Hydraulics Update Threshold= 0.02
Energy Slope Method= 1
Volume Change Method= 0
XS Weighting Method= 0
Number of US Weighted Cross Sections= 1
Number of DS Weighted Cross Sections= 1
Upstream XS Weight=0.25
Main XS Weight=0.5
Downstream XS Weight=0.25
Number of DS XS's Weighted with US Boundary= 1
Upstream Boundary Weight= 1
Weight of XSs Associated with US Boundary= 0
Number of US XS's Weighted with DS Boundary= 1
Downstream Boundary Weight= 0.5
Weight of XSs Associated with DS Boundary= 0.5
Sediment Output Level= 4
Mass or Volume Output= 0
Output Increment Type= 1
Profile and TS Output Increment= 10
XS Output Flag= 0
XS Output Increment= 10
Disregard all LS=0
Disregard all Conn=0
Disregard all Breaches=0
Disregard all Pumps=0

--- SALT BRANCH RAMIRENA CREEK.f01 (steady flow) ---

Flow Title=Multiple
Program Version=4.10
Number of Profiles= 7
Profile Names=10-year,25-year,50-year,1pct_min,100-year,1pct_plu,500-year
River Rch & RM=SALT BRANCH RAMI,Reach-1         ,54601
     173     239     293     266     359     486     547
River Rch & RM=SALT BRANCH RAMI,Reach-1         ,54052
     224     313     387     353     477     645     735
River Rch & RM=SALT BRANCH RAMI,Reach-1         ,51003
     355     506     635     585     791    1070    1250
River Rch & RM=SALT BRANCH RAMI,Reach-1         ,46026
     536     775     982     912    1233    1668    1979
River Rch & RM=SALT BRANCH RAMI,Reach-1         ,45622
     536     775     982     912    1233    1668    1979
River Rch & RM=SALT BRANCH RAMI,Reach-1         ,40472
     605     878    1114    1037    1403    1897    2260
River Rch & RM=SALT BRANCH RAMI,Reach-1         ,35365
     702    1023    1303    1215    1644    2223    2661
River Rch & RM=SALT BRANCH RAMI,Reach-1         ,30205
     723    1053    1339    1248    1688    2283    2726
River Rch & RM=SALT BRANCH RAMI,Reach-1         ,23012
     970    1427    1826    1712    2315    3131    3781
River Rch & RM=SALT BRANCH RAMI,Reach-1         ,18288
    1045    1538    1969    1846    2497    3376    4079
River Rch & RM=SALT BRANCH RAMI,Reach-1         ,17823
    1045    1538    1969    1846    2497    3376    4079
River Rch & RM=SALT BRANCH RAMI,Reach-1         ,12078
    1241    1836    2360    2219    3001    4059    4935
River Rch & RM=SALT BRANCH RAMI,Reach-1         ,10830
    1241    1836    2360    2219    3001    4059    4935
River Rch & RM=SALT BRANCH RAMI,Reach-1         ,7970
    1247    1844    2369    2226    3011    4072    4945
Boundary for River Rch & Prof#=SALT BRANCH RAMI,Reach-1         , 1
Up Type= 0
Dn Type= 3
Dn Slope=0.0027
Boundary for River Rch & Prof#=SALT BRANCH RAMI,Reach-1         , 2
Up Type= 0
Dn Type= 3
Dn Slope=0.0027
Boundary for River Rch & Prof#=SALT BRANCH RAMI,Reach-1         , 3
Up Type= 0
Dn Type= 3
Dn Slope=0.0027
Boundary for River Rch & Prof#=SALT BRANCH RAMI,Reach-1         , 4
Up Type= 0
Dn Type= 3
Dn Slope=0.0027
Boundary for River Rch & Prof#=SALT BRANCH RAMI,Reach-1         , 5
Up Type= 0
Dn Type= 3
Dn Slope=0.0027
Boundary for River Rch & Prof#=SALT BRANCH RAMI,Reach-1         , 6
Up Type= 0
Dn Type= 3
Dn Slope=0.0027
Boundary for River Rch & Prof#=SALT BRANCH RAMI,Reach-1         , 7
Up Type= 0
Dn Type= 3
Dn Slope=0.0027
DSS Import GetInterval= 0
DSS Import GetPeak= 0
DSS Import FillOption= 0

--- SALT BRANCH RAMIRENA CREEK.g01 (geometry) ---

Geom Title=Existing Conditions
Program Version=4.10

River Reach=SALT BRANCH RAMI,Reach-1
Reach XY= 30
      2188879.98     13245016.23      2191340.83     13244751.34
      2191969.66     13245810.07      2192637.12     13246060.22
      2194067.04     13245361.26      2196193.03     13246285.87
      2198708.43     13245845.21      2200215.73     13246917.08
      2201904.31     13246523.85      2202479.83     13247147.98
      2205582.98     13247726.41      2208236.86     13247649.61
      2208825.12     13248292.32      2209599.89      13248327.5
      2210923.41      13247251.8      2210909.06     13245200.89
       2212506.8     13243341.39      2212858.15     13240527.67
      2213201.91     13240204.75      2215047.45     13240406.85
      2216636.29      13238293.3      2215388.61      13234897.7
      2216379.37     13233940.15      2217647.79     13234213.32
      2219020.34     13233921.81       2219661.2     13232370.36
      2221012.69     13231829.52      2221320.93     13230593.41
      2222276.47     13230703.86      2222977.72     13230026.86

Type RM Length L Ch R = 1 ,54601   ,549,549,549
BEGIN DESCRIPTION:
SALT BRANCH RAMIRENA CREEK 69.0
END DESCRIPTION:
XS GIS Cut Line= 3
      2188987.72     13245646.87      2188937.72     13245046.85
      2188787.71     13244446.81
#Sta/Elev= 30
  4380.6  448.79  4400.7  448.36  4438.3  446.23  4450.9  446.29  4470.9  444.26
  4531.1  443.04  4551.2  441.27  4581.3  440.75  4601.4  439.47  4684.2  437.89
  4701.7  436.32  4731.8   435.3  4872.3   431.2  4902.4     431  4932.5  430.22
    4993  430.09  5000.5  428.96  5013.6  429.89  5147.6  430.87  5281.6  434.48
  5302.2  436.71  5335.7  437.01  5343.5  438.09    5395  438.52  5405.3  440.03
  5418.2  439.67  5436.2  443.41  5518.7   445.8  5541.9  448.59  5601.2  450.49
#Mann= 3 , 0 , 0
  4380.6      .1       0  4902.4    .035       0  5147.6      .1       0
Bank Sta=4902.4,5147.6
XS Rating Curve= 0 ,0
Exp/Cntr=0.3,0.1

Type RM Length L Ch R = 1 ,54052   ,469,469,469
BEGIN DESCRIPTION:
SALT BRANCH RAMIRENA CREEK 68.0
END DESCRIPTION:
XS GIS Cut Line= 3
      2189481.12     13245545.89      2189403.97      13244791.8
      2189254.73     13244351.54
#Sta/Elev= 30
  4436.4  443.34  4455.5  441.21  4519.9  440.19  4619.3  437.37  4626.4  436.32
  4666.6  435.33  4690.7   433.2    4737  431.73  4767.2  431.76  4787.3  430.61
  4818.1  430.35  4867.7  428.51  4948.1   427.2  4978.3  426.41  4988.1  425.48
  5068.7   427.3    5129  427.69  5284.1  431.23  5336.9  433.79  5368.6  434.25
  5384.8  435.73  5421.5  436.22  5463.6  438.88    5502  440.09  5558.7  442.26
  5573.3  443.08  5579.8  444.26  5611.4  444.52  5630.8   445.9  5659.3  446.36
#Mann= 5 ,-1 , 0
  4436.4      .1       0  4690.7     .05       0  4948.1    .035       0
  5068.7     .05       0    5502      .1       0
Bank Sta=4948.1,5068.7
XS Rating Curve= 0 ,0
Exp/Cntr=0.3,0.1

Type RM Length L Ch R = 1 ,53583   ,343,343,343
BEGIN DESCRIPTION:
SALT BRANCH RAMIRENA CREEK 67.0
END DESCRIPTION:
XS GIS Cut Line= 2
      2189949.03     13245700.22      2189774.89      13244471.3
#Sta/Elev= 30
  4377.6  445.38  4411.3  444.35  4490.5  440.19  4542.6  438.61  4552.7  437.66
  4632.4  434.28  4643.6  434.54  4694.1  431.55  4815.3  427.88  4835.5  426.67
  4875.9  426.33  4890.6  425.28  4946.6  424.33  4997.2  422.51  5027.4  424.03
  5057.7  423.53  5118.3  424.39  5300.1  428.29  5352.4   429.8  5360.7   430.6
  5411.2  431.36  5418.4  432.11  5423.4  431.56  5431.4  432.26  5441.5  431.94
  5522.3  435.06  5565.4  435.33  5603.1  437.57  5613.2  437.22  5618.8  438.05
#Mann= 5 ,-1 , 0
  4377.6     .05       0  4552.7      .1       0  4890.6     .05       0
  4946.6    .035       0  5118.3     .05       0
Bank Sta=4946.6,5118.3
XS Rating Curve= 0 ,0
Exp/Cntr=0.3,0.1

Type RM Length L Ch R = 1 ,53240   ,638,638,638
BEGIN DESCRIPTION:
SALT BRANCH RAMIRENA CREEK 66.0
END DESCRIPTION:
XS GIS Cut Line= 3
      2190137.72     13245796.85      2190187.72     13245046.85
      2190087.73     13244446.89
#Sta/Elev= 30
  4261.6  449.45  4281.6  449.09  4341.8  446.52  4381.9  444.28    4432  442.85
    4549  436.59  4622.4  434.23  4702.6     430  4722.6  429.72  4732.6  428.94
  4802.8  426.55  4852.9  425.68    4913  423.23  4943.1   422.4  4973.2  422.55
    5003  420.99  5010.8  421.76  5041.1   421.7  5094.4  423.18  5185.6  425.37
  5398.5   432.8    5510  437.48  5527.8  438.75  5532.8  438.31  5550.6  438.93
  5560.7  440.14    5581  440.67  5588.6  440.23  5601.3  441.33  5621.5  441.91
#Mann= 4 ,-1 , 0
  4261.6     .05       0    4549      .1       0    4913    .035       0
  5094.4     .05       0
Bank Sta=4913,5094.4
XS Rating Curve= 0 ,0
Exp/Cntr=0.3,0.1

Type RM Length L Ch R = 1 ,52602   ,647,647,647
BEGIN DESCRIPTION:
SALT BRANCH RAMIRENA CREEK 65.0
END DESCRIPTION:
XS GIS Cut Line= 3
      2190822.18     13245510.71      2190714.76     13244695.56
      2190354.58     13244348.02
#Sta/Elev= 30
  4399.9  443.28  4514.7  437.87  4524.8  436.73  4544.4  435.74  4595.4  433.69
  4605.5  432.67  4628.1  431.89  4635.8  430.86  4655.9  430.34  4701.6  428.02
  4736.6  427.24    4772  425.77  4858.9  422.25  4877.8   422.2  4887.9   421.5
  4958.5  420.18  4988.8  419.08  4998.6  418.12    5011  419.58  5039.2  419.27
  5069.5  420.07  5109.8   419.5  5180.4  419.55  5289.7  420.74  5296.9  421.38
  5303.9   421.1  5346.3     422  5445.4  425.04  5459.5  425.09  5722.6   434.4
#Mann= 4 ,-1 , 0
  4399.9     .05       0    4772      .1       0  4958.5    .035       0
  5069.5     .05       0
Bank Sta=4958.5,5069.5
XS Rating Curve= 0 ,0
Exp/Cntr=0.3,0.1

Type RM Length L Ch R = 1 ,51955   ,461,461,461
BEGIN DESCRIPTION:
SALT BRANCH RAMIRENA CREEK 64.0
END DESCRIPTION:
XS GIS Cut Line= 3
       2190887.7     13245546.89      2191337.72     13244746.85
       2191687.7     13244346.88
#Sta/Elev= 30
  4085.9  445.15  4277.5  438.16  4315.1  436.03  4579.3  427.55  4747.3   420.9
  4800.7  419.78  4812.3  420.18  4843.2  418.37  4871.6  417.97  4930.8  416.73
  4974.2  416.97  5000.7  415.53  5025.2  417.36  5039.4  417.01  5067.9  418.13
    5103  418.61  5117.2  419.69  5152.4  419.75  5174.2  421.25  5209.3   421.4
    5255  423.18  5277.7  424.66  5389.3  429.36    5401  430.91  5407.7  430.23
  5415.3  431.19  5493.1  434.74    5514  434.69  5521.6  435.79  5535.3  435.78
#Mann= 7 ,-1 , 0
  4085.9     .05       0  4800.7      .1       0  4871.6    .035       0
  5067.9      .1       0    5255     .08       0  5277.7      .1       0
  5389.3     .08       0
Bank Sta=4871.6,5067.9
XS Rating Curve= 0 ,0
Exp/Cntr=0.3,0.1

Type RM Length L Ch R = 1 ,51494   ,491,491,491
BEGIN DESCRIPTION:
SALT BRANCH RAMIRENA CREEK 63.0
END DESCRIPTION:
XS GIS Cut Line= 3
      2190937.71     13245546.86      2191687.72     13244996.85
      2192037.69     13244646.88
#Sta/Elev= 30
  4070.8  443.61    4099  443.84  4107.5  442.28  4128.3  441.46  4157.6  441.26
  4178.5  439.72  4184.7  440.61  4207.2  438.77    4285  436.83  4293.5  435.76
  4299.7  436.37  4314.3  434.87    4329  435.22  4393.2  432.16    4400  432.76
  4492.4  427.63  4506.5   428.3  4579.2  424.58  4639.5  423.02  4665.5  421.39
  4851.5  416.44  4997.5  414.44  5029.2  416.11  5128.1  418.57  5202.2  421.92
  5368.6  429.76  5425.1  434.03  5467.6  435.91  5481.7  438.01  5495.8  438.02
#Mann= 5 ,-1 , 0
  4070.8     .05       0  4639.5      .1       0  4851.5    .035       0
  5029.2     .08       0  5202.2      .1       0
Bank Sta=4851.5,5029.2
XS Rating Curve= 0 ,0
Exp/Cntr=0.3,0.1

Type RM Length L Ch R = 1 ,51003   ,323,323,323
BEGIN DESCRIPTION:
SALT BRANCH RAMIRENA CREEK 62.0
END DESCRIPTION:
XS GIS Cut Line= 3
      2191087.68     13245496.86      2191887.72     13245396.85
      2192287.76     13244996.82
#Sta/Elev= 30
  4187.2  437.88    4212   436.6    4276  433.93    4378  429.71  4499.7     424
  4519.8  424.26  4620.6  420.08  4779.4  416.17  4794.4  415.78    4870  413.84
  4943.1  413.47  4963.2   414.2    4997  413.39  5007.4  411.64  5021.8  413.26
  5120.7   415.5  5163.2  416.41  5177.3  417.25  5191.5  419.33  5205.6  417.85
  5275.8  421.79  5315.5  423.75    5347  424.51  5361.2  426.28  5403.6  427.73
  5431.9  429.87  5474.3  430.86  5488.4  432.94  5502.6  432.53  5559.2  435.48
#Mann= 9 ,-1 , 0
  4187.2     .05       0    4212      .1       0    4276     .05       0
    4378      .1       0  4779.4     .08       0  4794.4    .035       0
  5120.7      .1       0  5275.8     .08       0  5315.5     .05       0
Bank Sta=4794.4,5120.7
XS Rating Curve= 0 ,0
Exp/Cntr=0.3,0.1

Type RM Length L Ch R = 1 ,50680   ,655,655,655
BEGIN DESCRIPTION:
SALT BRANCH RAMIRENA CREEK 61.0
END DESCRIPTION:
XS GIS Cut Line= 4
      2191218.21      13246016.3      2191478.59     13245990.26
      2192285.88       13245413.      2192368.17      13245101.2
#Sta/Elev= 30
  4174.8  431.63    4320  426.13  4345.2  424.31  4415.5  422.16  4420.5   422.8
    4429   421.6  4481.9  419.52    4546  418.74  4553.1   417.5  4632.1   415.9
  4639.1  414.92  4653.9   414.6  4767.3  414.04  4804.2  413.29  4817.3  412.26
  4840.6  413.31  4897.2  412.38  4932.8  412.67  4962.3  411.75  4989.3  412.48
  5003.8  409.85  5012.7  411.57  5025.5  412.12  5184.7  413.05  5241.2  414.05
  5283.7   415.8  5333.8  416.96    5418  419.98  5471.1  422.11  5751.4  434.75
#Mann= 7 ,-1 , 0
  4174.8     .05       0    4429      .1       0  4632.1    .035       0
  5283.7      .1       0  5333.8     .05       0    5418     .08       0
  5471.1     .05       0
Bank Sta=4632.1,5283.7
XS Rating Curve= 0 ,0
Exp/Cntr=0.3,0.1

Type RM Length L Ch R = 1 ,50025   ,625,625,625
BEGIN DESCRIPTION:
SALT BRANCH RAMIRENA CREEK 60.0
END DESCRIPTION:
XS GIS Cut Line= 3
      2192437.72     13246696.81      2192387.72     13245996.85
      2192437.72     13245196.86
#Sta/Elev= 30
  4319.6  435.34  4359.7  434.04    4510  426.92  4540.1  425.09  4630.3  421.04
  4667.9  418.71  4680.5  418.81  4720.6  417.38  4730.6  416.23  4740.6  415.77
  4780.7   414.5  4800.8  413.34  4840.9  413.05    4881  411.22  4981.2  408.72
  5015.8  408.69  5018.6  408.19  5021.8  408.69  5051.4  408.75  5061.4  409.28
  5221.7  410.72    5342  413.46    5362  414.61  5412.1  415.65  5456.9  417.88
  5532.8  420.64  5592.5  423.66  5642.6  425.01  5762.8  429.93  5822.9  431.76
#Mann= 5 ,-1 , 0
  4319.6     .05       0  4740.6    .035       0  5412.1      .1       0
  5456.9     .08       0  5532.8     .05       0
Bank Sta=4740.6,5412.1
XS Rating Curve= 0 ,0
Exp/Cntr=0.3,0.1

Type RM Length L Ch R = 1 ,49400   ,357,357,357
BEGIN DESCRIPTION:
SALT BRANCH RAMIRENA CREEK 59.0
END DESCRIPTION:
XS GIS Cut Line= 3
      2193066.07     13246464.13       2192960.5     13245891.99
      2192728.93       13245262.
#Sta/Elev= 30
  4485.3  432.49  4553.7   427.9  4558.8  426.96  4594.4  425.17  4616.9  422.81
  4669.9   421.2  4685.9  419.71  4716.4  418.07  4727.9  416.79  4757.1  415.86
  4775.8  414.65  4828.3  413.52    4839  412.18  4868.9  411.26  4899.5  409.12
    4930  408.46  5011.1   403.6  5014.3   404.1  5083.2  404.96  5144.7  407.73
    5243  408.63    5275  410.02  5291.8  409.78  5392.2  411.21  5555.4  415.82
  5562.7  416.55  5573.3  416.53  5679.9   420.7  5702.4  422.29  5738.3  423.24
#Mann= 3 , 0 , 0
  4485.3     .05       0  4757.1    .035       0  5555.4     .05       0
Bank Sta=4757.1,5555.4
XS Rating Curve= 0 ,0
Exp/Cntr=0.3,0.1

Type RM Length L Ch R = 1 ,49043   ,89,89,89
BEGIN DESCRIPTION:
SALT BRANCH RAMIRENA CREEK 58.0
END DESCRIPTION:
XS GIS Cut Line= 4
      2193379.37     13246382.41      2193328.29     13245980.53
      2193161.42     13245442.46      2193022.48     13245042.58
#Sta/Elev= 30
    4349  429.89  4400.9  426.64  4405.9  426.97  4480.8  422.58  4586.5  417.81
  4606.6  415.51  4720.8  410.93  4773.3  409.99  4805.9  408.75  4811.1  408.07
  4908.9  405.46  4935.7  403.76  4938.9  404.26    4974  404.56    5077  404.27
  5124.4  404.78  5166.3  406.73  5187.2  408.47  5260.5  409.08  5277.8  409.88
  5418.7     413  5466.1  413.56  5528.3  415.67  5590.5  417.63  5609.2  417.53
  5621.6  418.46  5630.4   418.3  5693.9  420.26  5735.5  420.56  5740.8   421.4
#Mann= 3 , 0 , 0
    4349     .05       0  4606.6    .033       0  5528.3     .05       0
Bank Sta=4606.6,5528.3
XS Rating Curve= 0 ,0
Exp/Cntr=0.3,0.1

Type RM Length L Ch R = 1 ,48954   ,68,68,68
BEGIN DESCRIPTION:
Mapping XS 1ec1aad7
END DESCRIPTION:
XS GIS Cut Line= 4
      2193433.86     13246372.12      2193416.83     13246055.45
      2193249.96     13245326.68      2193032.36     13244905.08
#Sta/Elev= 30
  4338.8  429.14  4359.5  427.19  4574.4  416.83  4644.5  417.51  4672.1  416.67
  4763.1  416.04  4818.6  416.69  4848.9  415.86  4972.5   417.4  5030.9  416.31
    5036  417.04  5095.6  416.59  5121.8  414.67  5126.9  416.22  5146.9  416.53
  5198.2  415.27  5260.8  416.33  5298.6  415.58  5406.3  416.38  5470.9  414.12
  5619.2  417.64  5673.4  417.64  5740.9  419.78  5801.6  420.51  5819.7   421.1
  5829.5  419.98  5835.1  420.94  5842.2  420.17  5857.3  421.69    5878  422.09
#Mann= 4 ,-1 , 0
  4338.8     .05       0  4972.5     .03       0    5036     .05       0
  5801.6      .1       0
#XS Ineff= 2 , 0
       0 4950.75  417.65 5052.24       0  417.09
Permanent Ineff=
       T       T
Bank Sta=4972.5,5036
XS Rating Curve= 0 ,0
Exp/Cntr=0.3,0.1

Type RM Length L Ch R = 1 ,48886   ,854,854,854
BEGIN DESCRIPTION:
SALT BRANCH RAMIRENA CREEK 57.0
END DESCRIPTION:
XS GIS Cut Line= 4
      2193505.37      13246341.5      2193488.35     13246052.04
      2193294.23     13245227.92      2193172.16     13244956.65
#Sta/Elev= 30
  4351.3  425.29    4376  424.92  4416.1  423.14  4496.2  418.83  4636.3  412.54
  4687.7  411.98  4728.8  410.13  4739.1  410.39  4790.4  408.79  4801.2  409.28
  4821.2  408.32  4843.6  408.68  4903.4  407.54  4965.1  406.21  4985.6  406.94
  5006.2  406.41  5012.8  405.63  5018.2  406.69  5055.4  407.07  5060.5  407.74
  5129.4  407.46  5150.4  408.41  5211.6  408.46  5283.6   410.2  5446.9  411.72
  5562.6  415.13  5706.9  418.36  5712.4  419.14  5735.6  418.83  5785.4  420.15
#Mann= 3 , 0 , 0
  4351.3     .05       0  4903.4     .03       0  5060.5     .05       0
Bank Sta=4903.4,5060.5
XS Rating Curve= 0 ,0
Exp/Cntr=0.3,0.1

Type RM Length L Ch R = 1 ,48032   ,844,844,844
BEGIN DESCRIPTION:
Mapping XS d9a6ca15
END DESCRIPTION:
XS GIS Cut Line= 3
      2193302.06     13246544.56      2194088.51     13246028.95
      2194135.39     13244804.95
#Sta/Elev= 30
  3401.7  433.18    3492  433.32  3513.1  432.02  3585.4  430.87  3621.6  429.73
  3684.8  426.12  3779.1  423.54  3802.5  421.84  3844.6  421.19  3850.9  420.15
  3895.9  419.47  3901.9  418.19  3932.1  418.49  3938.1  417.31  4004.4  415.84
  4010.4   415.1  4031.5  415.52  4076.8  412.45  4257.5   407.7  4424.3   404.4
  4514.3  403.45  4845.4   403.1  4934.6  402.48  4984.7  401.15  4994.4  400.22
  5034.7  403.11  5069.6  404.97    5375  418.46  5493.7  425.23    5567  426.67
#Mann= 5 ,-1 , 0
  3401.7     .05       0  4845.4      .1       0  4934.6    .035       0
  5034.7      .1       0  5069.6     .05       0
Bank Sta=4934.6,5034.7
XS Rating Curve= 0 ,0
Exp/Cntr=0.3,0.1

Type RM Length L Ch R = 1 ,47188   ,514,514,514
BEGIN DESCRIPTION:
Mapping XS a1ce095a
END DESCRIPTION:
XS GIS Cut Line= 2
      2194479.16     13246221.63      2195609.34     13244815.41
#Sta/Elev= 30
  4437.4   416.3    4482  416.37  4518.5  415.27  4539.3  415.34  4553.7  414.49
  4560.1  414.98  4603.3  413.95  4617.7  412.72  4652.6  411.65  4675.9  410.78
  4802.8  405.63  4809.7   404.7  4866.9  402.89  4937.7  399.44  4952.1  399.28
  4980.6  397.58  4987.3  398.55  5022.5  398.11  5072.2  399.33  5193.7  399.26
  5321.7  400.11  5443.3  402.52  5585.3  407.58  5684.9  412.06  5833.7  420.91
  5862.5  421.96  6025.7  430.43  6054.5  431.13  6124.9  434.45  6241.5  437.92
#Mann= 5 ,-1 , 0
  4437.4     .05       0  4652.6     .08       0  4675.9     .05       0
  4952.1     .03       0  5072.2     .05       0
Bank Sta=4952.1,5072.2
XS Rating Curve= 0 ,0
Exp/Cntr=0.3,0.1

Type RM Length L Ch R = 1 ,46674   ,648,648,648
BEGIN DESCRIPTION:
Mapping XS b0e9dfef
END DESCRIPTION:
XS GIS Cut Line= 4
       2194691.7     13246210.35      2195138.47     13246139.81
      2195622.81     13245467.37      2195683.73     13245050.31
#Sta/Elev= 30
    4215  414.83  4322.3  412.14  4460.4  407.02  4534.9  405.36  4565.3  403.74
  4575.4  404.39  4585.3  403.57  4612.7  403.03  4630.5  402.36  4675.8   400.8
  4777.9  399.04  4918.8  397.68  4991.4  395.94  4998.3  395.24  5019.5  396.23
  5105.4  397.45    5206  398.62  5256.3  399.89  5262.5   400.6  5277.2  400.51
  5327.5   402.2  5442.9  407.29  5463.7   407.6  5493.2  409.79  5547.1   412.2
  5563.4  413.77  5587.5  414.73  5648.1  419.01  5749.2  424.27  5917.5  429.93
#Mann= 6 ,-1 , 0
    4215     .05       0  4612.7     .08       0  4630.5     .05       0
  4777.9      .1       0  4918.8     .03       0  5105.4     .05       0
Bank Sta=4918.8,5105.4
XS Rating Curve= 0 ,0
Exp/Cntr=0.3,0.1

Type RM Length L Ch R = 1 ,46026   ,404,404,404
BEGIN DESCRIPTION:
Mapping XS 3513bf7c
END DESCRIPTION:
XS GIS Cut Line= 3
      2195900.25     13247000.38      2195867.34     13246168.02
      2195881.44     13245147.62
#Sta/Elev= 30
  4186.1  412.71    4196  412.64  4279.7  410.04  4289.7  409.25  4319.7  408.98
  4369.8  407.51  4380.8  406.68    4650  398.72  4750.1  397.07  4800.1   395.6
  4860.1  394.85    4879  395.46  4910.2  395.36  4970.2  394.63    5000  393.08
  5010.3  393.86  5070.3  395.16  5100.3  394.69  5110.3   395.6  5300.3  396.09
  5390.3  397.81  5490.3  400.57  5580.3  403.62  5630.3  406.35  5740.3  410.69
  5810.3  411.76  5850.4  415.47  5880.4  415.75  5930.4  418.94  6039.6   423.1
#Mann= 4 ,-1 , 0
  4186.1     .08       0    4196     .05       0  4910.2     .04       0
  5110.3     .05       0
#XS Ineff= 2 , 0
         4879.07  395.47
Permanent Ineff=
       F       F
Bank Sta=4910.2,5110.3
XS Rating Curve= 0 ,0
Exp/Cntr=0.3,0.1

Type RM Length L Ch R = 1 ,45622   ,470,470,470
BEGIN DESCRIPTION:
SALT BRANCH RAMIRENA CREEK 56.0
END DESCRIPTION:
XS GIS Cut Line= 3
      2196637.72     13247046.85      2196237.72     13246246.85
      2196187.72     13245446.83
#Sta/Elev= 30
  4125.4  421.36  4315.6  413.73  4419.1  409.62  4474.8  408.03  4491.5  406.69
  4541.9  405.66  4550.2  404.55    4581  403.46    4595  404.02  4603.3  402.82
  4639.3  402.46  4653.7  401.63  4684.4  401.46  4692.8  400.53  4737.5  398.92
  4743.1  399.45  4751.5  398.46  4765.5  398.04  4930.4  394.89  5002.8  393.66
  5005.6  393.16    5017  394.13  5049.9  394.71  5180.1  394.74  5280.3  393.68
  5370.5  394.52  5583.4  400.33  5600.9  401.43  5731.2  405.96  5821.4  410.16
#Mann= 6 ,-1 , 0
  4125.4     .05       0  4315.6     .08       0  4419.1     .05       0
  4639.3      .1       0  4930.4     .04       0  5049.9     .05       0
Bank Sta=4930.4,5049.9
XS Rating Curve= 0 ,0
Exp/Cntr=0.3,0.1

Type RM Length L Ch R = 1 ,45152   ,434,434,434
BEGIN DESCRIPTION:
SALT BRANCH RAMIRENA CREEK 55.0
END DESCRIPTION:
XS GIS Cut Line= 3
      2196837.71     13246996.82      2196687.72     13246196.85
      2196287.73     13245396.88
#Sta/Elev= 30
  4194.3   420.8    4506  407.28  4540.1  405.83  4621.6  403.06  4651.3  401.41
  4656.3  401.56  4692.8  400.03  4733.5  399.56  4770.3  398.05    4814  396.09
  4871.7  394.43  4924.3  393.52  4967.5  392.14  4987.9  392.15  4997.8  391.01
  5005.7  391.95  5044.5   392.2  5052.9  393.09  5150.8  393.54  5284.9  392.87
  5335.2   393.5    5366  393.36  5455.4  395.02  5558.8  397.87  5611.9  400.22
    5693  402.82  5709.8  404.03  5813.2  407.74  5821.6   408.5  5902.6  412.08
#Mann= 6 ,-1 , 0
  4194.3     .05       0    4506     .08       0  4540.1     .05       0
  4770.3      .1       0  4924.3    .035       0  5052.9     .05       0
Bank Sta=4924.3,5052.9
XS Rating Curve= 0 ,0
Exp/Cntr=0.3,0.1

Type RM Length L Ch R = 1 ,44718   ,484,484,484
BEGIN DESCRIPTION:
SALT BRANCH RAMIRENA CREEK 54.0
END DESCRIPTION:
XS GIS Cut Line= 3
      2197237.72     13246546.85      2197087.72     13246146.85
      2196337.71     13245346.84
#Sta/Elev= 30
  4582.6  407.51  4622.4  405.82  4768.6  400.37  4774.8  399.05  4823.8  397.99
    4884  395.22    4903  393.74  4939.5  392.32  4956.4  391.21  4994.7  390.43
  4999.8  389.69  5007.1  390.47  5037.9  391.08  5045.2  392.12  5061.3  392.28
  5108.7  393.05  5122.9  392.88  5130.2  391.74    5137  391.64  5158.5  392.63
  5180.5  392.29  5321.2  391.55  5382.7  392.14  5434.5  392.52  5455.5  391.88
  5483.8  392.93  5646.5  395.91    5880  403.84  5979.1  408.44  6106.4  413.17
#Mann= 8 ,-1 , 0
  4582.6     .08       0  4622.4     .05       0    4884      .1       0
  4939.5    .035       0  5045.2      .1       0  5061.3     .05       0
  5180.5      .1       0  5382.7     .05       0
Bank Sta=4939.5,5045.2
XS Rating Curve= 0 ,0
Exp/Cntr=0.3,0.1

Type RM Length L Ch R = 1 ,44234   ,224,224,224
BEGIN DESCRIPTION:
SALT BRANCH RAMIRENA CREEK 53.0
END DESCRIPTION:
XS GIS Cut Line= 3
      2197337.73     13246546.82      2197487.72     13245946.85
      2197587.73     13245146.81
#Sta/Elev= 30
    4344  407.81  4378.6  406.85  4479.6  403.41  4573.3  399.83  4622.3  398.81
  4632.6  396.94  4655.8  396.55  4673.8  395.22  4691.9  395.85  4725.4  394.17
  4807.8  391.63  4820.7  391.95  4838.7  390.91    4880  390.54  4883.9  390.33
  4952.1  388.92  4982.6  389.15  5000.2  388.63    5005  387.85  5022.9  389.38
  5073.3  390.22  5083.7  390.28  5123.7  389.78  5182.9  390.26  5242.1  390.34
    5282  391.33  5415.9  393.89  5587.6  401.02  5635.2  402.94  5768.7  409.18
#Mann= 11 ,-1 , 0
    4344     .05       0  4378.6     .08       0  4479.6     .05       0
    4880     .08       0  4883.9    .035       0  5073.3     .08       0
  5083.7     .05       0  5182.9      .1       0    5282     .05       0
  5587.6     .08       0  5635.2     .05       0
Bank Sta=4880,5073.3
XS Rating Curve= 0 ,0
Exp/Cntr=0.3,0.1

Type RM Length L Ch R = 1 ,44010   ,105,105,105
BEGIN DESCRIPTION:
Mapping XS bb2b3c8d
END DESCRIPTION:
XS GIS Cut Line= 4
       2197357.6     13246584.52      2197690.94     13245893.53
      2197697.89     13245782.42      2197604.37     13245100.12
#Sta/Elev= 30
  4179.5  408.88  4257.1   406.4  4343.4  404.43  4365.2   403.4  4393.8  401.87
  4473.3  399.35  4576.6  396.31  4582.4  395.04    4621  394.38  4627.6  393.35
    4718  391.97  4723.6  391.26  4763.2  390.47  4827.6  389.96  4898.6  389.43
  4932.6  386.66  4963.4  387.08  4976.8  386.83  4983.2  385.94  4993.5  386.78
  5023.5  387.07  5134.3  386.69  5154.5  389.01  5169.7  389.74  5366.4  393.98
  5406.8  396.47  5447.2  397.77  5507.9  400.91  5689.9  408.34  5746.7   411.3
#Mann= 9 ,-1 , 0
  4179.5     .05       0  4257.1     .08       0  4365.2     .05       0
  4393.8     .08       0  4473.3     .05       0  4827.6     .08       0
  4898.6    .035       0  5169.7     .08       0  5507.9     .05       0
Bank Sta=4898.6,5169.7
XS Rating Curve= 0 ,0
Exp/Cntr=0.3,0.1

Type RM Length L Ch R = 1 ,43905   ,95,95,95
BEGIN DESCRIPTION:
Mapping XS 06d3e961
END DESCRIPTION:
XS GIS Cut Line= 5
      2197409.69     13246563.67      2197763.86     13245949.08
      2197805.53     13245837.97      2197798.58     13245751.17
      2197642.63     13245082.29
#Sta/Elev= 30
  4206.4   407.6  4296.7  405.45    4334  403.25  4392.9  402.95  4606.7  394.52
  4628.5  394.89  4650.1   393.3  4714.7  392.37  4745.2  390.66  4838.3  389.44
  4860.6  389.87  4869.9   391.1  4897.2  390.56  4928.8  393.64  4967.8  393.68
  4973.2  395.72  4992.7   395.2  5028.3  396.78  5065.1  398.36  5075.6  395.74
  5126.3  396.27  5144.3  393.91  5149.4  394.28    5192  387.79  5228.6  389.65
  5269.7  389.87  5324.8  391.51  5331.3  392.59  5444.2  395.57  5808.3  410.99
#Mann= 4 ,-1 , 0
  4206.4      .1       0  4973.2    .035       0  5028.3      .1       0
  5808.3     .05       0
#XS Ineff= 2 ,-1
 4492.43 4975.08  395.05 5068.77 5540.06   396.4
Permanent Ineff=
       T       T
Bank Sta=4973.2,5028.3
XS Rating Curve= 0 ,0
Exp/Cntr=0.3,0.1

Type RM Length L Ch R = 1 ,43810   ,446,446,446
BEGIN DESCRIPTION:
SALT BRANCH RAMIRENA CREEK 52.0
END DESCRIPTION:
XS GIS Cut Line= 3
      2197337.75     13246696.82      2197887.72     13245896.85
      2197687.72     13245096.85
#Sta/Elev= 30
  4037.8  411.62  4087.1  409.92  4268.3  405.76  4281.3  404.59    4332  402.26
  4361.8  403.14  4373.7  402.77  4491.1  398.67  4562.1  395.71  4723.9  391.95
  4756.2  391.79    4765  390.83    4786  390.37  4843.4  389.91  4850.8  389.55
  4929.4  388.75    5073  388.79  5109.1  388.08  5183.8   388.2    5225  389.36
  5232.8  387.03  5237.7  386.51    5256  388.25  5266.3  387.98  5297.2  389.53
  5340.9  390.75  5451.8  394.97  5521.4  396.85  5534.3  397.83  5833.2  409.92
#Mann= 8 ,-1 , 0
  4037.8     .05       0  4373.7     .08       0  4491.1     .05       0
  4723.9     .08       0  4843.4     .05       0  4850.8     .03       0
  5297.2      .1       0  5340.9     .05       0
Bank Sta=4850.8,5297.2
XS Rating Curve= 0 ,0
Exp/Cntr=0.3,0.1

Type RM Length L Ch R = 1 ,43364   ,402,402,402
BEGIN DESCRIPTION:
SALT BRANCH RAMIRENA CREEK 51.0
END DESCRIPTION:
XS GIS Cut Line= 3
      2197637.73     13246646.85      2198287.72     13245846.85
      2198587.74     13245446.83
#Sta/Elev= 30
  3945.5  403.81  4009.9  401.75  4066.2  400.64  4080.5  399.75    4194  397.09
  4251.5  395.01  4350.8  393.18  4542.4  390.24  4670.3  389.59    4699  388.97
  4705.7  389.68  4713.4  389.06  4734.2  389.68  4748.6  388.52  4777.3  388.44
  4783.7  387.83  4911.8  387.84    4973  386.12  4989.8  386.46  5004.1  385.08
  5012.7   386.6  5076.3     387  5133.6  388.23    5219  390.09    5319  393.84
  5326.3  394.69    5419  397.91  5448.1  399.45    5469  399.86  5476.3  400.57
#Mann= 4 ,-1 , 0
  3945.5     .05       0  4350.8     .08       0  4777.3     .03       0
  5133.6     .05       0
Bank Sta=4777.3,5133.6
XS Rating Curve= 0 ,0
Exp/Cntr=0.3,0.1

Type RM Length L Ch R = 1 ,42962   ,452,452,452
BEGIN DESCRIPTION:
SALT BRANCH RAMIRENA CREEK 50.0
END DESCRIPTION:
XS GIS Cut Line= 3
      2197487.69     13247046.88      2198687.72     13245846.85
      2198837.72     13245546.86
#Sta/Elev= 30
  3307.2  416.13  3434.5  411.18  3797.1  400.15  3830.5  399.28  3844.6  397.77
  3858.8   398.2  3940.3  396.41  4113.3  392.59    4283  391.01  4339.6  391.37
    4382  389.94  4576.1  387.34  4636.6  385.76  4711.7  385.64  4792.2  387.35
    4799  386.84  4806.3   386.3  4848.7  387.03  4905.3  386.67  4961.9  385.29
  4989.9  383.72  5040.6  385.38  5057.4  387.24  5095.9   389.4  5191.6  392.93
  5197.2  392.36  5213.9  394.07  5258.6   396.5  5286.6  397.19  5339.7  400.04
#Mann= 9 ,-1 , 0
  3307.2     .05       0  3797.1     .08       0  3940.3     .05       0
  4576.1      .1       0  4711.7     .08       0    4799      .1       0
  4905.3    .035       0  5057.4     .08       0  5095.9     .05       0
Bank Sta=4905.3,5057.4
XS Rating Curve= 0 ,0
Exp/Cntr=0.3,0.1

Type RM Length L Ch R = 1 ,42510   ,436,436,436
BEGIN DESCRIPTION:
SALT BRANCH RAMIRENA CREEK 49.0
END DESCRIPTION:
XS GIS Cut Line= 3
      2198487.75     13246846.82      2199087.72     13246046.85
      2199187.73     13245646.82
#Sta/Elev= 30
  3967.9  400.31  4304.3  388.24  4354.3  386.89  4389.7  387.11  4410.6  385.93
  4467.9  385.63  4543.5  385.53  4566.6  385.47  4654.3  384.77  4689.7  385.28
  4717.9  384.65    4746  385.39    4796  384.57  4816.2  385.02  4831.4  384.15
  4870.7  384.64  4939.7  384.61    4988  382.86  4990.8  382.36    4994  382.86
  5032.3  383.69  5068.4  386.07  5144.1  388.89  5184.3  390.24  5225.5  392.67
  5245.1  392.73  5274.5  393.12  5315.7  397.16  5346.2  398.12  5380.2  399.59
#Mann= 10 ,-1 , 0
  3967.9     .05       0  4543.5      .1       0  4566.6     .05       0
  4816.2      .1       0  4870.7     .05       0    4988     .03       0
    4994     .05       0  5144.1     .08       0  5245.1      .1       0
  5346.2     .08       0
Bank Sta=4467.9,5068.4
XS Rating Curve= 0 ,0
Exp/Cntr=0.3,0.1

Type RM Length L Ch R = 1 ,42074   ,844,844,844
BEGIN DESCRIPTION:
SALT BRANCH RAMIRENA CREEK 48.0
END DESCRIPTION:
XS GIS Cut Line= 3
      2198687.69     13246996.88      2199487.72     13246196.85
      2199987.72     13245396.86
#Sta/Elev= 30
  3863.7  399.64  4075.9  390.22  4217.3  385.79  4245.6  386.31    4288  384.52
  4344.6  384.89  4358.7  383.97  4556.7  383.52  4937.5  383.25  4988.6  381.41
  4991.3  380.91  4994.6  381.41  5060.6  383.65  5170.2  387.24  5337.1  389.04
  5484.8   393.5  5582.7  397.37  5669.1  402.15  5699.7   402.8  5705.6  403.85
  5749.8  405.12  5811.3  408.99  5830.6  410.34  5844.2  409.98  5857.7  407.82
  5879.5  408.23  5888.4  409.03  5903.1  412.95  5909.6  412.27  5938.5  414.43
#Mann= 7 ,-1 , 0
  3863.7     .05       0  4937.5      .1       0  4988.6     .07       0
  4994.6      .1       0  5484.8     .08       0  5582.7      .1       0
  5811.3     .05       0
Bank Sta=4556.7,5060.6
XS Rating Curve= 0 ,0
Exp/Cntr=0.3,0.1

Type RM Length L Ch R = 1 ,41230   ,446,446,446
BEGIN DESCRIPTION:
SALT BRANCH RAMIRENA CREEK 47.0
END DESCRIPTION:
XS GIS Cut Line= 3
      2199698.59     13247683.34      2199820.11     13247058.34
      2200063.16     13245478.53
#Sta/Elev= 30
  4101.4  405.25  4250.6  400.24  4278.2  400.16  4301.6  398.27  4422.8   395.3
  4729.4  388.82  4886.5  383.49  4962.2   380.3  4999.7  375.89  5002.4  375.39
  5005.7  375.89  5012.5   377.3  5018.1  378.84  5023.1  378.24  5053.3  379.79
  5117.2  379.78  5159.7  379.93  5439.6  382.76  5518.7   383.3  5650.2   385.1
  5719.5  387.06  5932.5  394.57  6034.7  399.06  6085.3   399.5  6095.4  401.32
  6106.8  402.04  6125.7   403.8  6196.5  406.06  6201.8  407.27  6336.5   412.8
#Mann= 11 ,-1 , 0
  4101.4      .1       0  4422.8     .05       0  4999.7     .03       0
  5005.7     .05       0  5012.5      .1       0  5117.2     .05       0
  5159.7      .1       0  5439.6     .05       0  5719.5      .1       0
  5932.5     .08       0  6106.8     .05       0
Bank Sta=4886.5,5518.7
XS Rating Curve= 0 ,0
Exp/Cntr=0.3,0.1

Type RM Length L Ch R = 1 ,40784   ,186,186,186
BEGIN DESCRIPTION:
SALT BRANCH RAMIRENA CREEK 46.0
END DESCRIPTION:
XS GIS Cut Line= 3
      2200337.72     13247546.85      2200287.72     13246946.85
      2200187.72     13245846.87
#Sta/Elev= 30
  4376.8  402.99  4467.1  397.58  4530.3   395.1  4657.8  388.43  4800.8  383.75
  4888.6  380.28  4930.2  380.12  4958.8  379.57  4968.8  377.81  4981.4  377.45
    4996   373.1  4998.7   372.6    5002   373.1  5028.1  375.95  5149.6  378.33
  5189.7  381.06  5199.8  383.36  5209.8  383.99    5250  383.06    5260  381.64
  5270.1  383.17  5280.1   383.1  5290.2   380.4  5300.2  379.58  5424.8  380.63
  5581.4  383.23  5626.1  384.42  5643.5  385.11  5812.3  389.02  6083.4  398.55
#Mann= 9 ,-1 , 0
  4376.8     .05       0  4530.3      .1       0  4930.2     .12       0
    4996     .07       0    5002     .12       0  5028.1      .1       0
  5424.8     .05       0  5626.1      .1       0  5643.5     .05       0
Bank Sta=4800.8,5581.4
XS Rating Curve= 0 ,0
Exp/Cntr=0.3,0.1

Type RM Length L Ch R = 1 ,40598   ,126,126,126
BEGIN DESCRIPTION:
Mapping XS a5e59eb4
END DESCRIPTION:
XS GIS Cut Line= 3
      2200461.78     13247647.04      2200479.14     13246428.25
      2200433.99     13245813.62
#Sta/Elev= 30
  4272.8  399.68    4393  399.06    4453  397.65    4593  390.69    4623  390.53
  4668.9     388    4773  383.27    4823  381.18    4863  385.29    4873  384.56
    4883  380.86    4903  375.67  4923.1  373.46  4954.3  372.28  5000.1  369.49
  5002.8  368.99  5006.1  369.49  5063.1  371.07    5115  374.45  5173.1  376.82
  5183.1  378.29  5193.1  383.78  5203.1  384.79  5223.1  379.01  5293.1  378.07
  5331.7  378.65  5583.8  383.21  6051.6  395.41    6105  396.72    6108  396.72
#Mann= 9 ,-1 , 0
  4272.8     .05       0  4668.9      .1       0  4954.3     .12       0
  5000.1     .07       0  5006.1     .12       0    5115      .1       0
  5331.7     .05       0  6051.6      .1       0    6105     .08       0
Bank Sta=4773,5583.8
XS Rating Curve= 0 ,0
Exp/Cntr=0.3,0.1

Type RM Length L Ch R = 1 ,40472   ,143,143,143
BEGIN DESCRIPTION:
Mapping XS 61c471d2
END DESCRIPTION:
XS GIS Cut Line= 3
      2200531.22     13247650.44      2200600.66     13246886.58
      2200611.08     13245824.04
#Sta/Elev= 30
  4264.6  399.47  4358.6  399.83  4408.8  398.48    4459  395.59  4489.1  395.09
  4723.7  384.39  4740.1  383.63  4840.6  379.67  4870.7  380.66  4890.8  382.07
  4900.8  383.79  4939.9  383.88  4944.9  382.38  4972.8  383.15    5001  383.52
  5101.3  384.14  5161.3   382.6  5191.3  378.56  5221.3  378.69  5248.3  377.92
  5251.1  377.42  5254.3  377.92  5282.9  378.02  5481.4  380.49  5621.4  383.33
  5821.4  387.79  5881.4  388.43  5921.4  390.32  6009.7   392.7  6094.2   395.5
#Mann= 8 ,-1 , 0
  4264.6     .05       0  4723.7      .1       0  4972.8     .12       0
    5001      .1       0  5248.3     .07       0  5254.3      .1       0
  5282.9     .05       0  6009.7      .1       0
Bank Sta=4740.1,5621.4
XS Rating Curve= 0 ,0
Exp/Cntr=0.3,0.1

Type RM Length L Ch R = 1 ,40329   ,481,481,481
BEGIN DESCRIPTION:
SALT BRANCH RAMIRENA CREEK 45.0
END DESCRIPTION:
XS GIS Cut Line= 3
      2200687.72     13247546.83      2200737.72     13246946.85
      2200837.72     13245746.87
#Sta/Elev= 30
  4376.8  399.22  4396.8  399.09  4416.9  397.17  4426.9  395.51  4439.5  394.78
    4447  393.75  4477.1  392.26  4554.9  390.06  4577.5   388.8  4607.6  388.49
    4738  383.12  4888.5  377.64  4976.3  376.36  5038.6  376.24  5041.3  375.74
  5044.6  376.24  5089.2  376.62  5129.4  378.62    5162   377.4  5179.5  378.31
  5219.7  377.25  5282.4  377.55  5560.9  380.66  5711.5  382.93  5721.4  383.13
  5764.1  383.64  5867.9   387.1  6052.6  393.65  6072.6  395.05    6183  399.68
#Mann= 5 ,-1 , 0
  4376.8     .05       0  5038.6     .03       0  5044.6     .05       0
  5711.5      .1       0  5867.9     .05       0
Bank Sta=4738,5721.4
XS Rating Curve= 0 ,0
Exp/Cntr=0.3,0.1

Type RM Length L Ch R = 1 ,39848   ,447,447,447
BEGIN DESCRIPTION:
SALT BRANCH RAMIRENA CREEK 44.0
END DESCRIPTION:
XS GIS Cut Line= 3
      2201487.71     13248046.82      2201187.72     13246846.85
      2200887.73     13245646.88
#Sta/Elev= 30
  3763.4  413.94  3856.1  409.36  3910.3  408.67    3918  407.86  3951.5  406.78
  3959.2  405.88  4041.7  402.66  4075.2  400.71  4350.9  389.64  4487.5  385.97
  4528.7  384.23    4588  383.18  4729.7  379.92  4812.2  378.91  5007.6  373.47
  5010.4  372.97  5013.6  373.47  5044.5  374.61  5113.7  375.95  5162.4   375.9
  5265.7  376.55  5278.6  376.03  5381.7  377.67  5484.8  378.27  5678.9  381.35
  5742.5  383.27  5839.2  387.16  5958.9  391.85  6149.2  400.66  6237.2  403.67
#Mann= 8 ,-1 , 0
  3763.4     .05       0  5007.6     .03       0  5013.6     .05       0
  5044.5      .1       0  5162.4     .05       0  5678.9      .1       0
  5839.2     .05       0  6149.2     .08       0
Bank Sta=4588,5742.5
XS Rating Curve= 0 ,0
Exp/Cntr=0.3,0.1

Type RM Length L Ch R = 1 ,39401   ,542,542,542
BEGIN DESCRIPTION:
SALT BRANCH RAMIRENA CREEK 43.0
END DESCRIPTION:
XS GIS Cut Line= 3
      2201637.72     13247746.85      2201537.72     13246546.85
      2201637.72     13245346.87
#Sta/Elev= 30
  3829.4  404.95  3949.8  401.23  3959.8  401.56    4000  399.59  4050.2  398.15
  4060.2  397.16  4110.4  396.27  4270.9  390.53  4541.9   383.1    4582  381.58
  4990.4  371.76  4993.2  371.26  4996.4  371.76  5063.7  373.66  5251.2  376.98
  5381.5  380.16  5457.5  381.56  5505.2  383.25  5565.4  385.09  5595.5  386.81
  5625.6  387.22  5716.1  391.47    5773  393.94  5813.7  396.07  5876.5  398.18
  5906.6  400.33  5976.8  403.92  6006.9  404.81  6097.2  409.84  6237.7  416.24
#Mann= 7 ,-1 , 0
  3829.4     .05       0  4990.4     .03       0  4996.4     .05       0
  5251.2      .1       0  5381.5     .05       0  5716.1      .1       0
    5773     .05       0
Bank Sta=4541.9,5505.2
XS Rating Curve= 0 ,0
Exp/Cntr=0.3,0.1

Type RM Length L Ch R = 1 ,38859   ,250,250,250
BEGIN DESCRIPTION:
SALT BRANCH RAMIRENA CREEK 42.0
END DESCRIPTION:
XS GIS Cut Line= 4
      2201694.78     13247354.59      2201882.26     13246802.56
      2202087.12     13246562.97      2202014.24     13245851.53
#Sta/Elev= 30
  4198.7  393.93  4223.1  392.66  4365.3  389.54  4460.3  385.36  4468.9  384.21
  4505.6  383.23  4523.7  382.79  4576.5  379.54  4817.6  371.89  4839.6  370.46
  4852.4  368.84    4886   363.9  4888.8   363.4    4892   363.9  5073.4   364.2
  5096.9  366.88  5103.1  368.54  5133.2  371.78  5139.2  373.15  5144.2  372.01
  5193.6  375.43  5263.9  377.44  5332.8  380.48  5344.3  379.99  5418.8  381.79
    5465  383.31  5505.2  386.87  5535.1   387.5  5699.4  392.01  5812.1  395.69
#Mann= 7 ,-1 , 0
  4198.7     .05       0  4852.4      .1       0    4886     .07       0
    4892      .1       0  5418.8     .05       0  5535.1      .1       0
  5699.4     .05       0
Bank Sta=4505.6,5465
XS Rating Curve= 0 ,0
Exp/Cntr=0.3,0.1

Type RM Length L Ch R = 1 ,38609   ,146,146,146
BEGIN DESCRIPTION:
Mapping XS 5f25c7bd
END DESCRIPTION:
XS GIS Cut Line= 6
      2201746.83     13247340.79      2201889.21     13247038.67
      2202059.35     13246983.11      2202236.43     13246767.83
      2202264.21     13246646.31      2202173.93     13245743.51
#Sta/Elev= 30
  4252.8  393.36  4445.1  386.95  4511.4  383.04  4546.1   381.2  4548.9   380.7
  4552.1   381.2  4571.9  382.92  4577.7  385.26  4680.3  389.39  4783.6  387.63
  4797.9  389.39  4833.1  388.69  4839.6   390.2    5066  390.41  5107.1  387.63
    5120  389.62  5171.4  387.64  5180.7  385.37    5229  385.43  5260.1  383.27
  5331.2  387.82  5361.7  386.07  5392.2  388.67  5443.1  386.72  5457.7  388.03
  5520.7  382.01  5633.9  382.71    5702  384.91  5983.4  392.19    6078  394.19
#Mann= 7 ,-1 , 0
  4252.8     .05       0  4546.1     .07       0  4552.1     .05       0
  4680.3      .1       0  5520.7     .05       0    5702     .08       0
  5983.4     .05       0
Bank Sta=4511.4,5633.9
XS Rating Curve= 0 ,0
Exp/Cntr=0.3,0.1

Type RM Length L Ch R = 1 ,38463   ,445,445,445
BEGIN DESCRIPTION:
SALT BRANCH RAMIRENA CREEK 41.0
END DESCRIPTION:
XS GIS Cut Line= 3
      2201837.73     13247296.85      2202237.72     13246896.85
      2203137.69     13245796.89
#Sta/Elev= 30
  4447.2  390.96  4546.2  387.01  4602.8   383.1  4758.3  377.01  4857.3  372.17
  4970.4  370.67  4995.7  369.47  4998.5  368.97  5001.7  369.47  5013.5  369.53
  5040.9  370.43  5098.3  370.46  5133.5   372.3  5240.4  373.97  5388.6  374.35
  5588.6  375.91  5765.9  380.62    5852  384.33  5872.8  386.03  5986.2  390.48
  6014.9  392.55  6035.8  392.94  6064.5  395.33  6099.2  396.48  6171.4  400.45
  6192.2  402.33  6295.8  407.65  6334.4  409.76  6430.5  412.81  6434.1  412.79
#Mann= 8 ,-1 , 0
  4447.2     .05       0  4995.7     .03       0  5001.7     .05       0
  5013.5      .1       0  5388.6     .05       0  6099.2     .08       0
  6295.8     .05       0  6430.5     .08       0
Bank Sta=4857.3,5133.5
XS Rating Curve= 0 ,0
Exp/Cntr=0.3,0.1

Type RM Length L Ch R = 1 ,38018   ,517,517,517
BEGIN DESCRIPTION:
SALT BRANCH RAMIRENA CREEK 40.0
END DESCRIPTION:
XS GIS Cut Line= 3
      2201987.72     13247546.85      2202587.72     13247146.85
      2203087.72     13245946.86
#Sta/Elev= 30
  4309.8   390.7  4338.3  389.21  4345.9  390.13  4359.4  388.56  4381.5  387.61
  4482.6  384.62  4518.6  382.59  4590.7  381.09  4670.4  377.56  4692.9  377.72
    4735  376.08  4742.5  376.63  4842.3   373.3  4945.3   370.6  5014.4  367.52
  5017.1  367.02  5020.4  367.52  5093.2  370.18  5193.4  370.75  5240.1  370.86
  5427.2  371.93  5536.3  372.65  5644.4  375.14  5730.1  377.03  5772.4  377.55
  5908.4  383.14  6166.4  396.85  6215.5  399.65  6233.4  401.43  6330.9  406.59
#Mann= 10 ,-1 , 0
  4309.8     .05       0  4381.5      .1       0  4842.3     .05       0
  5014.4     .03       0  5020.4     .05       0  5240.1      .1       0
  5427.2     .08       0  5644.4     .05       0  5730.1     .08       0
  6166.4     .05       0
Bank Sta=4945.3,5193.4
XS Rating Curve= 0 ,0
Exp/Cntr=0.3,0.1

Type RM Length L Ch R = 1 ,37501   ,503,503,503
BEGIN DESCRIPTION:
SALT BRANCH RAMIRENA CREEK 39.0
END DESCRIPTION:
XS GIS Cut Line= 3
      2201987.69     13248146.88      2203087.72     13247146.85
      2203187.72     13245946.86
#Sta/Elev= 30
  3528.8     398  3599.5  396.49  3635.3   393.5  3755.5  388.59  3914.3  385.01
  4045.4  381.58  4142.6  380.27  4201.5  379.95  4222.5     381  4244.1  380.07
  4364.4  379.72  4371.1   380.4  4427.9  379.15  4505.6   379.1  4517.3  377.79
  4569.5  376.84  4576.6  377.44  4590.7  376.19  4668.5  373.95  4888.1  369.44
  4998.6  365.53  5001.3  365.03  5004.6  365.53  5065.6  368.65  5135.9  368.86
  5396.8  370.76  5587.4  374.55    5748  381.32  5921.1     390  6219.6  407.73
#Mann= 6 ,-1 , 0
  3528.8     .05       0  3914.3      .1       0  4142.6     .08       0
  4517.3     .05       0  4998.6     .03       0  5004.6     .05       0
Bank Sta=4888.1,5135.9
XS Rating Curve= 0 ,0
Exp/Cntr=0.3,0.1

Type RM Length L Ch R = 1 ,36998   ,530,530,530
BEGIN DESCRIPTION:
SALT BRANCH RAMIRENA CREEK 38.0
END DESCRIPTION:
XS GIS Cut Line= 4
      2203544.21     13248384.81      2203537.09     13247708.12
      2203608.32     13246696.65      2203466.24     13246050.18
#Sta/Elev= 30
  3841.6  387.45  3899.6  386.03  4003.5  385.55  4159.6  383.08  4289.6  378.11
  4399.6  374.85  4439.6  372.82  4449.6     373  4516.5  370.63  4609.8  369.07
  4679.9   368.7  4870.5  367.32  4910.6  366.93  4997.8  364.34  5000.5  363.84
  5003.8  364.34    5071  367.65  5321.6  375.61  5529.7  379.09  5583.3  379.01
  5736.9  381.31  5743.4  381.98  5748.5  381.66  5841.1  384.24  5951.9  388.37
  6013.3  390.98  6021.3  391.88  6026.5  391.48  6054.3   392.5  6194.2   398.6
#Mann= 5 ,-1 , 0
  3841.6     .05       0  4003.5      .1       0  4679.9     .05       0
  4997.8     .03       0  5003.8     .05       0
Bank Sta=4870.5,5071
XS Rating Curve= 0 ,0
Exp/Cntr=0.3,0.1

Type RM Length L Ch R = 1 ,36468   ,381,381,381
BEGIN DESCRIPTION:
SALT BRANCH RAMIRENA CREEK 37.0
END DESCRIPTION:
XS GIS Cut Line= 4
      2203765.01     13248484.57      2203992.96     13247971.67
      2204135.42     13246967.33      2204234.96     13246711.37
#Sta/Elev= 30
  3805.6  386.97  3934.4  383.35    3967  381.25    4019  381.25  4047.8  379.58
  4065.5   380.1  4175.2  377.69  4192.8   377.9  4343.2  372.88  4366.5  371.31
  4436.9  369.72  4462.6  368.22  4553.5  366.66  4593.9  367.14  4614.1  366.17
  4644.2  366.21  4856.5  366.08  4947.4  364.88  4994.9  362.66  4997.7  362.16
  5000.9  362.66  5098.9  366.37  5250.4  372.92  5260.5  372.61  5364.3  376.39
  5454.1  380.07  5459.4  380.98  5624.3  386.49  5644.6  387.27  5655.9  387.67
#Mann= 6 ,-1 , 0
  3805.6      .1       0  4644.2     .05       0  4994.9     .03       0
  5000.9     .05       0  5624.3     .08       0  5644.6      .1       0
Bank Sta=4856.5,5098.9
XS Rating Curve= 0 ,0
Exp/Cntr=0.3,0.1
