--- UNT 003 IN RACR.prj (project) ---

Proj Title=UNT 003 IN RACR Base Level Engineering
Current Plan=p01
Default Exp/Contr=0.3,0.1
English Units
Geom File=g01
Flow File=f01
Plan File=p01
BEGIN DESCRIPTION:
UNT 003 IN RACR
END DESCRIPTION:

--- UNT 003 IN RACR.p01 (plan) ---

Plan Title=Multiple Run
Short Identifier=Multiple
Geom File=g01
Flow File=f01
Subcritical Flow
K Sum by GR= 0
Std Step Tol= 0.01
Critical Tol= 0.01
Num of Std Step Trials= 20
Max Error Tol= 0.3
Flow Tol Ratio= 0.001
Split Flow NTrial= 30
Split Flow Tol= 0.02
Split Flow Ratio= 0.02
Log Output Level= 0
Friction Slope Method= 1
Unsteady Friction Slope Method= 2
Unsteady Bridges Friction Slope Method= 1
Parabolic Critical Depth
Global Vel Dist=  1 , 1 , 1
Global Log Level= 0
CheckData=True
Encroach Param= -1, 0, 0, 0
BEGIN DESCRIPTION:
Multiple Run
END DESCRIPTION:

--- UNT 003 IN RACR.f01 (steady flow) ---

Flow Title=Multiple
Number of Profiles=7
Profile Names=10-year,25-year,50-year,1pct_min,100-year,1pct_plu,500-year
River Rch & RM= UNT 003 IN RACR,Reach-1,18606
     266     371     460     418     566     765     870
River Rch & RM= UNT 003 IN RACR,Reach-1,11779
     343     486     606     555     751    1016    1173
River Rch & RM= UNT 003 IN RACR,Reach-1,6260
     394     560     701     645     872    1179    1370
Boundary for River Rch & Prof#=UNT 003 IN RACR,Reach-1,1
Up Type=0
Dn Type=3
Dn Slope=0.005
Boundary for River Rch & Prof#=UNT 003 IN RACR,Reach-1,2
Up Type=0
Dn Type=3
Dn Slope=0.005
Boundary for River Rch & Prof#=UNT 003 IN RACR,Reach-1,3
Up Type=0
Dn Type=3
Dn Slope=0.005
Boundary for River Rch & Prof#=UNT 003 IN RACR,Reach-1,4
Up Type=0
Dn Type=3
Dn Slope=0.005
Boundary for River Rch & Prof#=UNT 003 IN RACR,Reach-1,5
Up Type=0
Dn Type=3
Dn Slope=0.005
Boundary for River Rch & Prof#=UNT 003 IN RACR,Reach-1,6
Up Type=0
Dn Type=3
Dn Slope=0.005
Boundary for River Rch & Prof#=UNT 003 IN RACR,Reach-1,7
Up Type=0
Dn Type=3
Dn Slope=0.005

--- UNT 003 IN RACR.g01 (geometry) ---

Geom Title=Existing Conditions

River Reach=UNT 003 IN RACR,Reach-1
Reach XY= 30
      2196347.72     13240566.85      2196649.06     13240943.56
      2197237.56     13241099.10      2197873.12     13241072.50
      2198264.36     13241493.07      2198360.72     13241464.02
      2199253.85     13242086.91      2199959.05     13242830.31
      2200408.84     13243053.51      2202561.89     13242964.53
      2203389.13     13242657.28      2204345.02     13242754.20
      2204888.65     13242370.81      2205332.62     13242425.27
      2205957.72     13242306.86      2206205.25     13241942.46
      2206666.45     13241853.72      2207393.96     13241456.80
      2207946.62     13241699.40      2208275.37     13242051.14
      2208656.67     13242139.39      2208964.62     13242432.96
      2209873.67     13242708.77      2209973.19     13242840.85
      2210497.50     13242925.05      2210925.02     13243289.63
      2211293.94     13243356.91      2211571.72     13243139.89
      2211806.09     13243172.45      2212389.84     13243520.19

Type RM Length L Ch R = 1,18606,449,449,449
BEGIN DESCRIPTION:
UNT 003 IN RACR 40.0
END DESCRIPTION:
XS GIS Cut Line= 3
      2196037.70     13241146.88      2196437.72     13240746.85
      2196837.70     13240396.87
#Sta/Elev= 30
  4423.1  427.44  4564.6  423.14  4790.8  415.43  4895.6  412.82  4932.3  412.33
  4960.5  410.63  4974.7  410.76  4985.3  409.76  4992.9  409.63  4995.7  409.13
  4998.9  409.63  5052.9  411.30  5067.1  411.05  5081.4  411.53  5095.1  411.41
  5102.2  411.87  5108.9  411.48  5145.0  411.89  5201.4  413.04  5208.5  413.77
  5257.9  414.85  5378.4  419.19  5392.7  420.26  5427.8  421.18  5442.0  422.52
  5463.9  422.84  5478.1  423.97  5492.3  423.96  5499.0  424.66  5520.3  424.71
#Mann=4,-1,0
  4423.1    0.05       0  4895.6     0.1       0  4992.9    0.07       0
  4998.9     0.1       0
Bank Sta=4992.9,4998.9
Exp/Cntr=0.3,0.1

Type RM Length L Ch R = 1,18157,495,495,495
BEGIN DESCRIPTION:
UNT 003 IN RACR 39.0
END DESCRIPTION:
XS GIS Cut Line= 3
      2197137.72     13241796.86      2196787.72     13240996.85
      2196837.72     13240446.84
#Sta/Elev= 30
  4105.8  433.11  4110.2  433.09  4143.6  432.10  4204.0  427.82  4265.7  424.96
  4280.4  424.62  4289.4  423.44  4294.9  423.92  4312.8  421.96  4341.6  421.57
  4347.1  420.33  4365.0  420.50  4370.5  419.45  4378.7  420.90  4411.4  418.89
  4440.7  418.74  4446.1  417.91  4595.7  412.81  4662.1  411.30  4858.9  409.08
  4871.0  409.75  4970.0  409.60  4996.1  408.23  4998.8  407.73  5002.1  408.23
  5089.5  409.63  5250.1  413.78  5270.2  415.38  5300.3  415.76  5531.3  423.93
#Mann=6,-1,0
  4105.8    0.05       0  4110.2    0.08       0  4265.7    0.05       0
  4595.7     0.1       0  4996.1    0.07       0  5002.1     0.1       0
Bank Sta=4996.1,5002.1
Exp/Cntr=0.3,0.1

Type RM Length L Ch R = 1,17662,391,391,391
BEGIN DESCRIPTION:
UNT 003 IN RACR 38.0
END DESCRIPTION:
XS GIS Cut Line= 3
      2197264.77     13241599.67      2197180.24     13240669.90
      2196960.47     13240450.14
#Sta/Elev= 30
  4489.5  425.78  4499.5  425.20  4509.7  424.75  4514.8  425.36  4542.5  422.41
  4582.7  420.15  4602.8  420.23  4620.2  418.98  4625.2  419.38  4653.0  417.36
  4715.3  415.07  4841.1  409.71  4873.9  409.30  4924.1  407.36  5001.4  406.51
  5004.2  406.01  5007.4  406.51  5104.8  406.80  5282.9  409.06  5428.4  412.19
  5455.3  413.02  5462.4  414.35  5476.5  413.68  5568.5  416.78  5639.2  417.79
  5646.2  418.59  5660.4  418.57  5681.6  420.41  5724.0  420.70  5733.9  421.52
#Mann=5,-1,0
  4489.5    0.08       0  4499.5    0.05       0  4715.3     0.1       0
  5001.4    0.07       0  5007.4     0.1       0
Bank Sta=5001.4,5007.4
Exp/Cntr=0.3,0.1

Type RM Length L Ch R = 1,17271,445,445,445
BEGIN DESCRIPTION:
UNT 003 IN RACR 37.0
END DESCRIPTION:
XS GIS Cut Line= 3
      2197337.71     13241796.89      2197587.72     13240996.85
      2197987.74     13240596.84
#Sta/Elev= 30
  4221.4  433.64  4335.1  427.96  4431.0  424.29  4483.4  421.09  4502.7  421.13
  4535.2  418.70  4540.5  419.51  4555.6  418.49  4578.2  416.87  4588.1  417.24
  4658.1  414.25  4682.4  413.33  4702.8  411.45  4708.1  411.85  4755.8  410.30
  4778.3  408.69  4787.2  409.06  4797.7  408.11  4842.6  407.13  4892.0  405.83
  5017.7  405.12  5035.1  404.04  5037.9  403.54  5041.1  404.04  5043.3  404.81
  5172.7  405.59  5300.0  407.91  5455.6  413.35  5582.8  419.78  5625.3  420.78
#Mann=6,-1,0
  4221.4    0.05       0  4555.6    0.08       0  4658.1    0.05       0
  4842.6     0.1       0  5035.1    0.07       0  5041.1     0.1       0
Bank Sta=5035.1,5041.1
Exp/Cntr=0.3,0.1

Type RM Length L Ch R = 1,16826,242,242,242
BEGIN DESCRIPTION:
UNT 003 IN RACR 36.0
END DESCRIPTION:
XS GIS Cut Line= 3
      2197443.45     13241814.29      2198016.38     13241076.43
      2198250.74     13240447.13
#Sta/Elev= 30
  4177.2  432.34  4263.2  429.02  4599.0  413.02  4642.4  411.43  4648.8  412.41
  4655.1  410.73  4715.3  408.56  4755.6  407.40  4837.4  405.19  4922.1  403.39
  4959.6  403.03  4990.9  404.21  4997.3  400.55  5002.4  400.37  5005.2  399.87
  5008.4  400.37  5026.2  402.83  5112.0  405.31  5251.9  410.06  5385.2  415.27
  5409.7  417.33  5440.6  417.59  5569.8  422.86  5633.8  425.95  5647.6  427.62
  5655.1  426.97  5687.2  430.43  5702.9  430.46  5708.5  431.49  5782.9  434.53
#Mann=10,-1,0
  4177.2    0.05       0  4715.3     0.1       0  4755.6    0.05       0
  4837.4     0.1       0  4922.1    0.05       0  4959.6     0.1       0
  5002.4    0.07       0  5008.4     0.1       0  5112.0    0.08       0
  5251.9     0.1       0
Bank Sta=5002.4,5008.4
Exp/Cntr=0.3,0.1

Type RM Length L Ch R = 1,16584,76,76,76
BEGIN DESCRIPTION:
Mapping XS 8253f9e5
END DESCRIPTION:
XS GIS Cut Line= 4
      2197510.33     13241901.05      2198176.97     13241279.55
      2198385.30     13240567.75      2198385.30     13240551.13
#Sta/Elev= 30
  4190.2  434.33  4268.9  431.58  4559.1  418.19  4651.5  413.36  4679.3  410.50
  4821.0  409.35  4835.2  408.63  4842.5  406.37  4848.3  406.57  4856.6  404.20
  4863.5  403.71  4884.5  407.11  4891.8  406.70  4898.7  403.95  4906.0  403.10
  4934.3  402.29  4983.7  397.48  5030.5  397.21  5033.3  396.71  5036.5  397.21
  5061.6  399.89  5068.7  402.04  5089.7  405.37  5166.0  405.10  5281.6  405.52
  5332.1  409.93  5370.0  411.10  5692.4  422.95  5698.3  423.85  5859.9  427.36
#Mann=6,-1,0
  4190.2    0.05       0  4848.3     0.1       0  5030.5    0.07       0
  5036.5     0.1       0  5166.0    0.05       0  5370.0     0.1       0
Bank Sta=5030.5,5036.5
Exp/Cntr=0.3,0.1

Type RM Length L Ch R = 1,16508,81,81,81
BEGIN DESCRIPTION:
Mapping XS ea9b6ca7
END DESCRIPTION:
XS GIS Cut Line= 3
      2197538.08     13241973.99      2198242.94     13241321.22
      2198468.64     13240515.63
#Sta/Elev= 30
  4156.7  436.84  4657.0  414.32  4663.8  412.36  4692.1  410.58  4819.7  409.55
  4841.5  405.26  4859.2  403.02  4862.0  402.52  4865.2  403.02  4883.2  405.49
  4890.5  403.71  4904.7  404.55  4911.5  407.10  4933.1  406.53  4939.9  408.28
  4954.1  405.84  4960.9  407.50  4968.2  405.37  4975.0  407.61  4996.6  406.52
  5017.6  407.91  5045.9  406.96  5067.4  403.92  5134.3  404.40  5277.7  404.30
  5336.9  406.36  5371.0  410.74  5407.4  411.67  5651.6  420.72  5954.0  425.99
#Mann=6,-1,0
  4156.7    0.05       0  4841.5     0.1       0  4859.2    0.07       0
  4865.2     0.1       0  5134.3    0.05       0  5407.4     0.1       0
Bank Sta=4859.2,4865.2
Exp/Cntr=0.3,0.1

Type RM Length L Ch R = 1,16427,396,396,396
BEGIN DESCRIPTION:
Mapping XS 2156136e
END DESCRIPTION:
XS GIS Cut Line= 3
      2197590.13     13242033.05      2198357.52     13241324.69
      2198614.45     13240501.82
#Sta/Elev= 30
  4145.2  438.09  4480.7  422.75  4629.3  414.69  4643.4  414.89  4664.4  413.20
  4671.8  413.72  4678.6  412.44  4881.1  404.56  5022.6  401.66  5025.4  401.16
  5028.6  401.66  5053.7  402.11  5081.8  403.92  5129.3  403.92  5197.8  403.23
  5250.2  403.93  5270.0  404.26  5275.2  405.38  5292.0  406.23  5345.4  407.33
  5372.7  409.46  5470.1  413.18  5585.4  414.77  5643.1  416.79  5713.3  416.84
  5843.3  420.01  5848.5  419.19  5899.7  420.85  5908.2  420.10  6051.6  424.06
#Mann=6,-1,0
  4145.2    0.05       0  4881.1     0.1       0  5022.6    0.07       0
  5028.6     0.1       0  5129.3    0.05       0  5250.2     0.1       0
Bank Sta=5022.6,5028.6
Exp/Cntr=0.3,0.1

Type RM Length L Ch R = 1,16031,188,188,188
BEGIN DESCRIPTION:
UNT 003 IN RACR 35.0
END DESCRIPTION:
XS GIS Cut Line= 4
      2198024.16     13242123.34      2198732.52     13241380.25
      2198947.80     13240633.72      2199012.41     13240511.30
#Sta/Elev= 30
  4322.2  426.60  4357.7  425.38  4364.6  424.56  4513.1  417.38  4534.5  416.85
  4633.6  411.42  4711.3  408.09  4725.4  408.30  4739.6  406.98  4824.5  403.67
  4873.9  402.00  4987.1  400.34  5036.5  400.77  5083.2  400.21  5085.9  399.71
  5089.2  400.21  5334.0  403.43  5542.3  407.66  5563.6  408.14  5672.1  410.17
  5856.0  415.74  5956.0  419.95  5976.8  420.19  6018.4  422.34  6060.1  422.90
  6068.3  424.15  6121.5  426.81  6154.1  427.34  6225.8  431.23  6264.2  432.57
#Mann=6,-1,0
  4322.2    0.05       0  5083.2    0.03       0  5089.2    0.05       0
  5334.0     0.1       0  5542.3    0.05       0  5563.6     0.1       0
Bank Sta=5083.2,5089.2
Exp/Cntr=0.3,0.1

Type RM Length L Ch R = 1,15843,419,419,419
BEGIN DESCRIPTION:
UNT 003 IN RACR 34.0
END DESCRIPTION:
XS GIS Cut Line= 3
      2198237.70     13242146.87      2198637.72     13241746.85
      2199187.74     13240996.83
#Sta/Elev= 30
  4421.8  419.18  4464.3  416.81  4520.8  414.97  4775.4  404.22  4902.7  400.76
  4973.4  399.75  4998.0  398.77  5000.8  398.27  5004.0  398.77  5024.2  399.32
  5066.8  399.11  5216.4  400.81  5287.4  403.40  5387.7  405.92  5396.2  406.57
  5417.0  406.55  5481.9  408.46  5488.1  409.54  5495.9  409.06  5644.8  413.75
  5653.2  415.03  5667.9  414.68  5718.0  416.83  5753.5  417.61  5768.2  419.13
  5803.7  420.27  5818.4  421.60  5839.2  421.37  5904.0  423.47  5917.6  424.42
#Mann=4,-1,0
  4421.8    0.05       0  4998.0    0.03       0  5004.0    0.05       0
  5066.8     0.1       0
Bank Sta=4998,5004
Exp/Cntr=0.3,0.1

Type RM Length L Ch R = 1,15424,517,517,517
BEGIN DESCRIPTION:
UNT 003 IN RACR 33.0
END DESCRIPTION:
XS GIS Cut Line= 3
      2198637.75     13242346.82      2198987.72     13241946.85
      2199187.72     13241146.84
#Sta/Elev= 30
  4447.6  415.45  4610.3  409.97  4716.6  404.80  4738.5  404.69  4769.3  403.45
  4808.7  402.41  4844.8  400.45  4929.2  398.26  5002.3  397.05  5010.0  398.02
  5030.6  398.07  5068.8  396.90  5071.6  396.40  5074.8  396.90  5144.0  398.19
  5154.3  399.00  5195.5  399.69  5244.5  401.77  5360.4  404.59  5368.2  405.81
  5381.1  405.29  5414.6  407.49  5455.8  408.73  5484.1  410.54  5497.0  410.49
  5525.4  411.98  5698.0  417.35  5752.1  418.11  5785.6  420.41  5803.7  420.44
#Mann=4,-1,0
  4447.6    0.05       0  4769.3     0.1       0  5068.8    0.07       0
  5074.8     0.1       0
Bank Sta=5068.8,5074.8
Exp/Cntr=0.3,0.1

Type RM Length L Ch R = 1,14907,419,419,419
BEGIN DESCRIPTION:
UNT 003 IN RACR 32.0
END DESCRIPTION:
XS GIS Cut Line= 2
      2198972.16     13242613.93      2199799.21     13241820.64
#Sta/Elev= 30
  4433.3  410.43  4527.0  407.62  4535.2  406.87  4583.6  406.18  4590.9  405.53
  4640.2  405.23  4647.5  404.40  4781.7  399.67  4845.3  398.09  4859.4  398.60
  4909.1  396.68  4986.8  395.51  4994.0  394.67  5005.2  394.51  5007.9  394.01
  5011.2  394.51  5029.2  396.05  5050.6  395.19  5100.0  395.62  5156.6  396.37
  5163.5  396.95  5184.9  396.71  5276.8  398.88  5333.4  400.67  5347.5  401.77
  5368.9  401.83  5375.8  402.71  5404.1  404.01  5446.6  405.03  5579.3  410.99
#Mann=4,-1,0
  4433.3    0.05       0  4535.2     0.1       0  5005.2    0.07       0
  5011.2     0.1       0
Bank Sta=5005.2,5011.2
Exp/Cntr=0.3,0.1

Type RM Length L Ch R = 1,14488,441,441,441
BEGIN DESCRIPTION:
UNT 003 IN RACR 31.0
END DESCRIPTION:
XS GIS Cut Line= 3
      2199287.74     13242846.84      2199687.72     13242496.85
      2200087.73     13242196.85
#Sta/Elev= 30
  4444.2  410.91  4494.0  408.91  4514.9  407.33  4550.5  406.69  4592.7  404.19
  4628.8  403.33  4678.1  400.79  4713.3  400.06  4735.9  398.90  4841.4  395.28
  4951.3  393.22  4954.1  392.72  4957.3  393.22  4983.0  394.02  4989.2  393.43
  5018.4  393.76  5168.4  398.50  5183.0  399.51  5203.8  399.69  5212.1  400.71
  5233.0  400.99  5262.1  402.83  5283.0  403.08  5333.0  405.34  5362.1  407.36
  5375.7  408.88  5418.4  410.30  5439.2  410.20  5472.9  412.34  5475.7  412.34
#Mann=5,-1,0
  4444.2    0.05       0  4735.9     0.1       0  4951.3    0.07       0
  4957.3     0.1       0  5472.9    0.05       0
Bank Sta=4951.3,4957.3
Exp/Cntr=0.3,0.1

Type RM Length L Ch R = 1,14047,178,178,178
BEGIN DESCRIPTION:
UNT 003 IN RACR 30.0
END DESCRIPTION:
XS GIS Cut Line= 3
      2199415.71     13243318.59      2200049.36     13242745.70
      2200192.20     13242200.32
#Sta/Elev= 30
  4269.4  417.37  4364.3  412.85  4463.0  409.83  4696.9  400.51  4746.2  397.80
  4767.8  398.72  4810.4  395.03  4859.8  395.44  4888.1  399.43  4894.9  399.46
  4923.3  394.57  4930.7  392.37  4937.5  388.86  4965.9  382.75  5026.4  382.40
  5029.1  381.90  5032.4  382.40  5043.6  383.45  5051.0  385.70  5057.8  386.48
  5072.0  391.88  5079.4  393.59  5100.4  397.88  5114.6  399.40  5132.2  399.29
  5184.5  395.23  5218.2  397.57  5293.9  399.64  5308.5  401.21  5687.4  417.96
#Mann=3,-1,0
  4269.4    0.05       0  5026.4    0.03       0  5032.4    0.05       0
Bank Sta=5026.4,5032.4
Exp/Cntr=0.3,0.1

Type RM Length L Ch R = 1,13869,160,160,160
BEGIN DESCRIPTION:
UNT 003 IN RACR 29.0
END DESCRIPTION:
XS GIS Cut Line= 3
      2199606.66     13243409.75      2200144.85     13242884.59
      2200262.01     13242181.65
#Sta/Elev= 30
  4294.8  415.21  4375.4  412.86  4615.9  403.18  4686.6  398.83  4707.7  399.30
  4729.0  397.84  4736.0  396.06  4750.2  395.33  4827.9  395.21  4853.2  393.56
  4855.9  393.06  4859.2  393.56  4891.6  395.58  4898.6  397.47  4955.2  399.01
  5074.9  398.64  5092.4  397.50  5097.4  395.87  5115.4  394.00  5153.2  395.12
  5166.1  396.44  5186.4  395.09  5214.0  397.63  5267.5  399.05  5348.6  402.96
  5358.7  402.37  5368.9  403.64  5439.8  406.48  5518.2  410.89  5759.4  421.43
#Mann=3,-1,0
  4294.8    0.05       0  4853.2    0.03       0  4859.2    0.05       0
Bank Sta=4853.2,4859.2
Exp/Cntr=0.3,0.1

Type RM Length L Ch R = 1,13709,377,377,377
BEGIN DESCRIPTION:
Mapping XS 109f9dfa
END DESCRIPTION:
XS GIS Cut Line= 3
      2199762.88     13243540.00      2200327.14     13242901.95
      2200383.56     13242307.38
#Sta/Elev= 30
  4254.8  415.44  4274.3  415.52  4472.6  406.69  4579.4  403.13  4600.6  401.45
  4621.5  401.47  4643.2  400.56  4657.5  398.97  4678.4  400.00  4699.5  398.60
  4763.7  396.38  4784.6  396.54  4869.9  393.39  4898.4  393.42  4987.4  390.76
  4990.1  390.26  4993.4  390.76  5121.7  393.05  5182.0  395.00  5202.1  397.05
  5212.1  395.21  5222.2  395.27  5232.2  397.24  5362.8  402.25  5423.1  405.68
  5433.1  404.87  5443.2  406.47  5480.8  408.39  5573.7  411.93  5703.8  418.30
#Mann=3,-1,0
  4254.8    0.05       0  4987.4    0.03       0  4993.4    0.05       0
Bank Sta=4987.4,4993.4
Exp/Cntr=0.3,0.1

Type RM Length L Ch R = 1,13332,378,378,378
BEGIN DESCRIPTION:
UNT 003 IN RACR 28.0
END DESCRIPTION:
XS GIS Cut Line= 3
      2200478.98     13243652.08      2200614.61     13243266.04
      2200578.10     13242306.21
#Sta/Elev= 30
  4391.5  415.61  4471.2  411.12  4481.8  411.46  4490.2  410.43  4526.5  409.21
  4534.8  408.20  4557.5  407.78  4651.4  403.16  4662.0  403.39  4693.8  399.78
  4707.1  399.56  4715.0  400.82  4732.8  399.15  4847.7  394.30  4997.0  389.67
  4999.8  389.17  5003.0  389.67  5114.3  391.11  5200.2  394.31  5240.2  395.00
  5248.6  395.84  5260.2  396.83  5280.2  395.20  5300.2  397.87  5322.8  398.63
  5630.5  411.93  5637.5  413.05  5642.5  412.65  5710.5  415.81  5761.2  417.12
#Mann=5,-1,0
  4391.5    0.05       0  4997.0    0.03       0  5003.0    0.05       0
  5248.6     0.1       0  5322.8    0.05       0
Bank Sta=4997,5003
Exp/Cntr=0.3,0.1

Type RM Length L Ch R = 1,12954,549,549,549
BEGIN DESCRIPTION:
UNT 003 IN RACR 27.0
END DESCRIPTION:
XS GIS Cut Line= 2
      2201076.19     13243960.74      2200867.17     13242000.95
#Sta/Elev= 30
  4081.1  413.83  4105.1  413.41  4117.0  414.11  4135.3  412.25  4175.5  410.56
  4306.8  407.08  4349.5  404.57  4366.6  403.58  4394.2  403.80  4447.0  400.27
  4461.9  401.19  4768.8  391.46  4997.2  388.23  4999.9  387.73  5003.2  388.23
  5030.3  388.99  5089.3  388.68  5177.0  391.12  5261.6  393.47  5291.8  395.21
  5322.0  395.22  5352.1  397.56  5372.3  396.10  5402.4  398.87  5563.3  404.15
  5593.5  404.10  5643.8  406.79  5663.9  406.46  5925.4  412.26  6052.0  413.48
#Mann=7,-1,0
  4081.1    0.05       0  4349.5     0.1       0  4461.9    0.05       0
  4997.2    0.03       0  5003.2    0.05       0  5089.3     0.1       0
  5177.0    0.05       0
Bank Sta=4997.2,5003.2
Exp/Cntr=0.3,0.1

Type RM Length L Ch R = 1,12405,382,382,382
BEGIN DESCRIPTION:
Mapping XS 9dd94a3b
END DESCRIPTION:
XS GIS Cut Line= 3
      2201659.04     13244148.82      2201659.04     13243302.44
      2201019.45     13242120.82
#Sta/Elev= 30
  3874.4  422.09  3996.4  419.58  4246.4  411.29  4441.6  402.27  4442.8  402.21
  4546.4  398.13  4566.4  399.11  4586.4  396.58  4686.4  393.63  4733.4  391.21
  4909.1  386.62  4977.3  386.47  4981.6  385.66  4984.3  385.16  4987.6  385.66
  5102.4  386.82  5175.8  386.06  5191.9  387.11  5213.8  386.14  5425.8  388.92
  5487.6  389.89  5703.5  395.43  5716.3  395.66  5781.7  398.63  5787.4  396.91
  5803.6  397.12  5825.4  397.93  5831.1  399.64  5841.5  400.03  6064.4  406.68
#Mann=9,-1,0
  3874.4    0.05       0  4441.6    0.08       0  4442.8    0.05       0
  4981.6    0.03       0  4987.6    0.05       0  5425.8     0.1       0
  5487.6    0.05       0  5703.5     0.1       0  5716.3    0.05       0
Bank Sta=4981.6,4987.6
Exp/Cntr=0.3,0.1

Type RM Length L Ch R = 1,12023,244,244,244
BEGIN DESCRIPTION:
UNT 003 IN RACR 26.0
END DESCRIPTION:
XS GIS Cut Line= 4
      2202367.32     13243907.69      2201981.29     13243172.15
      2201710.04     13242707.89      2201089.66     13241691.31
#Sta/Elev= 30
  4024.0  404.56  4033.4  404.57  4146.8  401.71  4288.6  397.84  4313.3  396.76
  4341.2  397.13  4373.5  395.50  4486.9  392.17  4488.4  392.14  4660.5  389.76
  4803.6  386.09  4933.6  385.71  4996.8  383.69  4999.5  383.19  5002.8  383.69
  5008.0  384.54  5242.8  384.68  5335.7  386.85  5439.4  387.33  5526.7  388.28
  5592.6  389.05  5619.1  390.48  5644.6  390.70  5762.6  392.82  5880.5  394.19
  5978.3  395.51  6116.3  397.26  6157.9  398.00  6442.6  402.98  6583.3  406.56
#Mann=18,-1,0
  4024.0    0.08       0  4033.4     0.1       0  4146.8    0.08       0
  4288.6    0.05       0  4373.5    0.08       0  4486.9     0.1       0
  4488.4    0.08       0  4996.8    0.07       0  5002.8    0.08       0
  5439.4     0.1       0  5526.7    0.08       0  5619.1    0.05       0
  5644.6    0.08       0  5762.6     0.1       0  5880.5    0.08       0
  5978.3     0.1       0  6116.3    0.08       0  6157.9     0.1       0
Bank Sta=4996.8,5002.8
Exp/Cntr=0.3,0.1

Type RM Length L Ch R = 1,11779,538,538,538
BEGIN DESCRIPTION:
UNT 003 IN RACR 25.0
END DESCRIPTION:
XS GIS Cut Line= 3
      2202528.99     13243771.99      2201845.67     13242431.43
      2201756.99     13242076.71
#Sta/Elev= 30
  4118.1  407.05  4192.4  404.70  4305.0  400.13  4307.9  399.84  4417.7  395.94
  4512.0  392.29  4530.3  391.85  4642.9  387.65  4703.2  385.73  4731.0  386.19
  4747.6  384.85  4885.5  383.13  4980.8  381.96  4992.2  382.31  4996.3  381.27
  4999.1  380.77  5002.3  381.27  5124.5  383.04  5201.4  383.01  5318.6  385.69
  5328.6  385.90  5482.0  391.35  5492.4  392.68  5498.0  391.85  5543.9  393.16
  5653.5  397.14  5798.7  402.44  5803.9  401.45  5858.7  402.92  5988.4  406.75
#Mann=18,-1,0
  4118.1     0.1       0  4192.4    0.08       0  4305.0    0.05       0
  4307.9     0.1       0  4417.7    0.08       0  4512.0     0.1       0
  4530.3    0.08       0  4642.9    0.05       0  4885.5    0.08       0
  4980.8    0.05       0  4996.3    0.04       0  5002.3    0.05       0
  5124.5    0.08       0  5318.6     0.1       0  5328.6    0.08       0
  5543.9     0.1       0  5653.5    0.08       0  5858.7    0.05       0
Bank Sta=4996.3,5002.3
Exp/Cntr=0.3,0.1

Type RM Length L Ch R = 1,11241,384,384,384
BEGIN DESCRIPTION:
UNT 003 IN RACR 24.0
END DESCRIPTION:
XS GIS Cut Line= 3
      2202701.14     13243761.56      2202664.63     13243140.85
      2202628.17     13242130.39
#Sta/Elev= 30
  4186.4  405.67  4328.1  400.95  4341.4  401.13  4365.7  399.46  4431.5  397.97
  4469.2  396.11  4631.9  389.93  4651.9  390.01  4673.7  388.55  4702.0  388.60
  4712.0  387.64  4807.7  384.29  4902.2  382.21  4922.3  380.98  4952.3  380.78
  4972.3  379.38  5049.3  378.69  5052.1  378.19  5055.3  378.69  5096.2  379.27
  5142.9  380.68  5194.0  380.73  5272.5  382.02  5345.2  384.37  5602.7  394.60
  5612.7  395.73  5642.7  396.17  5747.5  400.58  5803.1  402.66  5819.3  402.75
#Mann=10,-1,0
  4186.4    0.05       0  4365.7     0.1       0  4469.2    0.05       0
  5049.3    0.03       0  5055.3    0.05       0  5096.2     0.1       0
  5194.0    0.05       0  5345.2     0.1       0  5747.5    0.05       0
  5803.1     0.1       0
Bank Sta=5049.3,5055.3
Exp/Cntr=0.3,0.1

Type RM Length L Ch R = 1,10857,402,402,402
BEGIN DESCRIPTION:
UNT 003 IN RACR 23.0
END DESCRIPTION:
XS GIS Cut Line= 4
      2203102.80     13243735.50      2203087.15     13243239.96
      2202925.44     13242358.40      2202779.41     13242102.84
#Sta/Elev= 30
  4075.3  395.67  4101.9  395.37  4134.0  395.33  4154.0  393.72  4214.0  391.59
  4334.1  387.53  4344.1  388.28  4406.9  385.98  4592.6  381.09  4703.9  379.26
  4848.7  378.50  4873.5  379.54  4899.6  378.08  4926.6  379.02  4950.4  377.99
  4970.8  378.41  4998.3  376.54  5001.0  376.04  5004.3  376.54  5043.0  378.52
  5147.2  380.07  5245.3  383.50  5318.8  387.49  5346.9  387.91  5448.6  393.22
  5458.8  393.07  5581.2  398.64  5603.5  399.75  5619.3  401.08  5761.7  404.94
#Mann=8,-1,0
  4075.3    0.05       0  4101.9     0.1       0  4406.9    0.05       0
  4998.3    0.03       0  5004.3    0.05       0  5147.2     0.1       0
  5581.2    0.05       0  5603.5     0.1       0
Bank Sta=4998.3,5004.3
Exp/Cntr=0.3,0.1

Type RM Length L Ch R = 1,10455,515,515,515
BEGIN DESCRIPTION:
UNT 003 IN RACR 22.0
END DESCRIPTION:
XS GIS Cut Line= 4
      2203582.70     13243662.48      2203546.19     13243239.96
      2203280.16     13242405.35      2203021.07     13242270.62
#Sta/Elev= 30
  3968.7  392.93  4024.5  390.53  4064.7  389.73  4082.4  388.34  4087.2  388.73
  4124.9  387.32  4134.9  387.92  4145.0  386.70  4185.1  385.16  4313.8  381.37
  4318.8  381.81  4375.8  379.43  4427.5  378.84  4467.2  377.44  4574.5  376.40
  4815.9  376.61  4857.9  375.97  4941.8  376.55  5001.8  375.31  5004.6  374.81
  5007.8  375.31  5078.3  378.37  5120.3  378.98  5151.7  380.55  5204.2  381.07
  5348.9  385.30  5373.0  386.83  5431.5  388.30  5463.1  390.51  5560.8  394.04
#Mann=5,-1,0
  3968.7     0.1       0  4082.4    0.05       0  5001.8    0.03       0
  5007.8    0.05       0  5348.9     0.1       0
Bank Sta=5001.8,5007.8
Exp/Cntr=0.3,0.1

Type RM Length L Ch R = 1,9940,424,424,424
BEGIN DESCRIPTION:
UNT 003 IN RACR 21.0
END DESCRIPTION:
XS GIS Cut Line= 3
      2204198.13     13243552.04      2203905.14     13243052.87
      2203807.48     13242173.98
#Sta/Elev= 30
  4074.0  394.49  4091.6  394.45  4205.0  389.85  4224.0  388.74  4276.8  387.76
  4282.6  386.71  4298.3  387.05  4325.5  385.45  4437.0  381.50  4590.2  377.37
  4819.8  373.89  4920.5  373.94  4940.6  373.05  4946.0  373.91  4959.4  373.81
  4997.9  372.69  5000.7  372.19  5003.9  372.69  5011.0  374.07  5051.3  374.60
  5147.3  378.40  5212.2  380.43  5222.7  381.58  5256.8  382.28  5343.0  385.35
  5363.2  385.23  5398.8  387.26  5473.8  389.11  5514.1  391.07  5537.1  391.10
#Mann=7,-1,0
  4074.0     0.1       0  4205.0    0.05       0  4959.4     0.1       0
  4997.9    0.07       0  5003.9     0.1       0  5147.3    0.05       0
  5256.8     0.1       0
Bank Sta=4997.9,5003.9
Exp/Cntr=0.3,0.1

Type RM Length L Ch R = 1,9516,478,478,478
BEGIN DESCRIPTION:
UNT 003 IN RACR 20.0
END DESCRIPTION:
XS GIS Cut Line= 4
      2204380.80     13243260.85      2204354.72     13242973.93
      2204177.36     13242441.86      2204042.22     13242166.37
#Sta/Elev= 30
  4479.1  389.19  4513.2  388.87  4553.4  386.79  4563.4  387.32  4583.5  385.54
  4678.9  382.47  4683.9  381.75  4771.5  378.23  4785.2  378.74  4848.4  375.67
  4903.2  374.20  4929.6  372.77  4943.3  372.83  4974.9  371.33  4985.5  372.11
  4989.8  371.06  4992.6  370.56  4995.8  371.06  5007.4  371.30  5057.6  371.99
  5124.6  372.21  5190.2  373.54  5295.4  376.19  5382.1  378.85  5411.9  379.71
  5422.7  381.04  5496.3  383.11  5524.4  385.20  5623.2  387.95  5634.9  389.09
#Mann=8,-1,0
  4479.1    0.05       0  4989.8    0.03       0  4995.8    0.05       0
  5007.4     0.1       0  5057.6    0.05       0  5190.2     0.1       0
  5295.4    0.05       0  5382.1     0.1       0
Bank Sta=4989.8,4995.8
Exp/Cntr=0.3,0.1

Type RM Length L Ch R = 1,9038,107,107,107
BEGIN DESCRIPTION:
UNT 003 IN RACR 19.0
END DESCRIPTION:
XS GIS Cut Line= 3
      2204487.71     13243246.89      2204687.72     13242546.85
      2204287.75     13242146.88
#Sta/Elev= 30
  4269.4  389.11  4364.3  385.34  4398.1  384.95  4437.1  382.54  4543.7  379.95
  4611.3  376.71  4684.1  375.69  4695.8  374.58  4792.2  372.28  4841.4  371.28
  4883.0  373.94  4893.4  371.16  4902.5  370.15  4907.7  372.22  4941.5  366.34
  4946.7  367.35  4955.8  365.79  4984.0  364.42  4986.8  363.92  4990.0  364.42
  5025.7  364.91  5039.9  367.37  5054.0  372.29  5068.2  374.19  5082.3  373.51
  5096.4  371.00  5157.8  371.34  5365.1  374.72  5505.4  379.51  5563.1  381.58
#Mann=6,-1,0
  4269.4    0.05       0  4792.2     0.1       0  4984.0    0.07       0
  4990.0     0.1       0  5157.8    0.05       0  5505.4     0.1       0
Bank Sta=4984,4990
Exp/Cntr=0.3,0.1

Type RM Length L Ch R = 1,8931,111,111,111
BEGIN DESCRIPTION:
Mapping XS 32ecbe38
END DESCRIPTION:
XS GIS Cut Line= 4
      2204575.40     13243149.36      2204811.52     13242566.01
      2204738.60     13242427.12      2204433.06     13241677.16
#Sta/Elev= 30
  4257.0  384.75  4551.0  374.55  4675.7  371.60  4741.2  370.83  4874.6  370.39
  4919.2  371.67  4925.8  368.83  4938.8  368.52  4941.6  368.02  4944.8  368.52
  4964.3  369.70  4969.9  371.32  4975.7  374.08  4986.3  374.89  4992.0  372.88
  4998.3  373.93  5020.9  370.34  5030.4  371.19  5036.1  372.72  5046.0  371.70
  5053.8  370.08  5065.1  370.05  5194.5  372.35  5379.9  376.53  5594.2  380.88
  5612.9  381.99  5680.6  383.10  5695.8  384.12  5725.3  383.92  5853.0  387.73
#Mann=6,-1,0
  4257.0    0.05       0  4741.2     0.1       0  4938.8    0.07       0
  4944.8     0.1       0  5194.5    0.05       0  5379.9     0.1       0
Bank Sta=4938.8,4944.8
Exp/Cntr=0.3,0.1

Type RM Length L Ch R = 1,8820,151,151,151
BEGIN DESCRIPTION:
Mapping XS 83190cff
END DESCRIPTION:
XS GIS Cut Line= 3
      2204610.13     13243170.18      2204863.60     13242527.82
      2204742.40     13241817.95
#Sta/Elev= 30
  4174.4  385.34  4236.5  382.52  4253.2  382.45  4290.6  380.40  4320.4  379.46
  4339.2  379.61  4374.5  377.42  4446.7  375.28  4597.2  371.43  4712.6  370.41
  4812.8  370.37  4823.0  369.85  4876.1  370.63  4977.5  368.95  4990.9  369.36
  4994.8  368.61  4997.6  368.11  5000.8  368.61  5146.7  373.65  5262.0  377.41
  5302.2  378.41  5312.3  379.91  5322.4  379.64  5383.3  382.05  5413.7  382.41
  5423.9  383.30  5515.2  385.36  5522.0  386.32  5582.2  388.55  5585.1  387.77
#Mann=6,-1,0
  4174.4    0.05       0  4712.6     0.1       0  4994.8    0.07       0
  5000.8     0.1       0  5146.7    0.05       0  5262.0     0.1       0
Bank Sta=4994.8,5000.8
Exp/Cntr=0.3,0.1

Type RM Length L Ch R = 1,8669,255,255,255
BEGIN DESCRIPTION:
UNT 003 IN RACR 18.0
END DESCRIPTION:
XS GIS Cut Line= 3
      2204637.72     13243196.87      2204987.72     13242396.85
      2204937.73     13241996.89
#Sta/Elev= 30
  4105.6  385.18  4149.3  383.51  4160.2  384.15  4182.0  382.03  4190.2  381.69
  4195.7  382.59  4219.1  380.77  4236.6  380.60  4271.3  378.72  4334.8  377.49
  4356.7  376.29  4498.6  372.24  4591.7  370.52  4736.8  369.81  4795.2  369.84
  4818.6  370.51  4847.8  369.46  4912.2  369.40  4996.0  368.04  4998.7  367.54
  5002.0  368.04  5029.2  368.72  5156.0  374.71  5279.6  379.68  5311.4  381.63
  5331.5  382.07  5339.1  382.95  5344.1  382.74  5361.8  384.24  5381.9  384.68
#Mann=6,-1,0
  4105.6    0.05       0  4736.8     0.1       0  4996.0    0.07       0
  5002.0     0.1       0  5156.0    0.05       0  5279.6     0.1       0
Bank Sta=4996,5002
Exp/Cntr=0.3,0.1

Type RM Length L Ch R = 1,8414,286,286,286
BEGIN DESCRIPTION:
Mapping XS 89754dc4
END DESCRIPTION:
XS GIS Cut Line= 3
      2205471.00     13243229.48      2205189.33     13242259.29
      2205012.36     13241993.83
#Sta/Elev= 30
  4127.3  385.76  4171.7  383.94  4202.9  381.86  4228.8  381.83  4255.0  380.57
  4269.5  380.73  4301.2  378.67  4432.0  373.85  4473.7  371.78  4551.6  369.88
  4585.2  368.46  4640.3  367.36  4681.9  367.60  4804.3  366.18  4807.1  365.68
  4810.3  366.18  4817.3  366.82  4894.4  367.31  4941.6  368.16  4952.7  367.34
  5004.7  367.17  5131.2  371.95  5205.1  373.95  5226.1  375.81  5248.6  375.81
  5262.2  376.81  5313.2  377.66  5364.6  380.12  5428.9  382.40  5456.6  384.12
#Mann=7,-1,0
  4127.3    0.08       0  4269.5    0.05       0  4804.3    0.07       0
  4810.3    0.05       0  4894.4     0.1       0  5131.2    0.05       0
  5364.6     0.1       0
Bank Sta=4804.3,4810.3
Exp/Cntr=0.3,0.1

Type RM Length L Ch R = 1,8128,476,476,476
BEGIN DESCRIPTION:
UNT 003 IN RACR 17.0
END DESCRIPTION:
XS GIS Cut Line= 3
      2206287.70     13243146.83      2205487.72     13242396.85
      2205087.75     13241996.88
#Sta/Elev= 30
  3916.8  391.32  3923.9  390.36  3952.2  388.96  3966.3  389.92  3983.2  388.41
  4010.3  387.43  4334.2  376.08  4362.7  374.57  4503.6  370.10  4602.8  366.32
  4638.5  366.35  4652.6  365.41  4730.3  364.13  4822.1  365.77  4914.4  366.23
  4928.6  366.50  4935.5  367.48  4940.3  367.09  4985.3  366.37  4992.1  365.41
  4996.4  363.98  4999.2  363.48  5002.4  363.98  5006.3  366.43  5069.9  367.28
  5098.2  366.92  5195.8  369.05  5338.6  372.96  5502.5  379.13  5579.0  381.97
#Mann=10,-1,0
  3916.8     0.1       0  3983.2    0.05       0  4010.3     0.1       0
  4362.7    0.08       0  4503.6    0.05       0  4940.3     0.1       0
  4996.4    0.07       0  5002.4     0.1       0  5195.8    0.05       0
  5502.5     0.1       0
Bank Sta=4996.4,5002.4
Exp/Cntr=0.3,0.1

Type RM Length L Ch R = 1,7652,495,495,495
BEGIN DESCRIPTION:
UNT 003 IN RACR 16.0
END DESCRIPTION:
XS GIS Cut Line= 3
      2206237.72     13242696.86      2205937.72     13242296.85
      2205137.73     13241596.87
#Sta/Elev= 30
  4514.8  380.43  4578.3  377.68  4601.3  377.33  4614.8  376.24  4664.8  374.85
  4722.0  371.85  4732.1  371.58  4778.3  370.37  4848.9  367.02  4892.9  364.73
  5004.5  361.52  5007.3  361.02  5010.5  361.52  5011.7  362.77  5149.1  363.26
  5156.7  363.82  5238.1  364.44  5319.9  365.45  5375.9  365.16  5510.7  367.82
  5638.9  372.58  5723.3  377.37  5837.2  381.83  5863.7  383.83  5929.3  386.71
  5943.5  387.95  5950.2  387.66  6021.3  392.39  6035.6  392.29  6077.8  394.80
#Mann=8,-1,0
  4514.8    0.05       0  4722.0    0.08       0  4732.1    0.05       0
  4848.9     0.1       0  5004.5    0.07       0  5010.5     0.1       0
  5238.1    0.05       0  5863.7     0.1       0
Bank Sta=5004.5,5010.5
Exp/Cntr=0.3,0.1

Type RM Length L Ch R = 1,7157,465,465,465
BEGIN DESCRIPTION:
UNT 003 IN RACR 15.0
END DESCRIPTION:
XS GIS Cut Line= 3
      2206637.73     13242746.88      2206237.72     13241946.85
      2206237.72     13241196.81
#Sta/Elev= 30
  4094.9  389.34  4184.4  384.94  4237.5  383.65  4256.3  382.49  4310.1  380.81
  4318.5  379.80  4326.9  380.05  4349.3  378.38  4407.8  375.77  4452.7  374.53
  4483.4  372.73  4606.7  367.99  4658.3  365.57  4690.3  365.40  4788.1  362.43
  4891.6  361.38  4899.9  361.72  4991.9  359.67  4996.4  358.21  4999.1  357.71
  5002.4  358.21  5019.4  360.06  5079.0  361.38  5149.4  364.39  5199.4  364.85
  5209.4  365.79  5409.4  372.78  5588.3  381.34  5619.4  382.26  5739.4  388.44
#Mann=10,-1,0
  4094.9    0.05       0  4256.3     0.1       0  4407.8    0.05       0
  4606.7    0.08       0  4658.3    0.05       0  4891.6     0.1       0
  4996.4    0.07       0  5002.4     0.1       0  5079.0    0.05       0
  5588.3     0.1       0
Bank Sta=4996.4,5002.4
Exp/Cntr=0.3,0.1

Type RM Length L Ch R = 1,6692,432,432,432
BEGIN DESCRIPTION:
UNT 003 IN RACR 14.0
END DESCRIPTION:
XS GIS Cut Line= 3
      2206737.72     13242646.89      2206687.72     13241846.85
      2206487.73     13241446.87
#Sta/Elev= 30
  4194.9  386.09  4233.2  384.61  4265.1  383.18  4272.6  382.27  4305.2  381.54
  4385.3  378.06  4415.4  377.47  4425.4  376.25  4524.0  372.42  4555.6  371.49
  4593.2  369.25  4598.2  369.55  4615.8  368.23  4695.9  366.32  4788.0  362.91
  4876.3  361.17  4887.2  360.33  4926.4  359.23  4946.4  360.15  4966.4  358.36
  4976.5  358.53  5001.9  356.94  5004.6  356.44  5007.9  356.94  5041.2  359.21
  5085.9  359.55  5165.3  362.68  5242.5  365.12  5278.8  367.24  5443.7  373.98
#Mann=8,-1,0
  4194.9    0.05       0  4233.2     0.1       0  4524.0    0.05       0
  4788.0    0.08       0  4887.2     0.1       0  5001.9    0.07       0
  5007.9     0.1       0  5165.3    0.05       0
Bank Sta=5001.9,5007.9
Exp/Cntr=0.3,0.1

Type RM Length L Ch R = 1,6260,425,425,425
BEGIN DESCRIPTION:
UNT 003 IN RACR 13.0
END DESCRIPTION:
XS GIS Cut Line= 3
      2206987.72     13242346.90      2207037.72     13241596.85
      2206637.72     13241196.85
#Sta/Elev= 30
  4221.2  375.16  4301.4  372.04  4311.4  372.19  4341.5  370.45  4401.6  368.82
  4411.7  369.05  4572.0  364.01  4662.2  362.50  4682.3  361.55  4712.3  361.40
  4722.4  360.77  4752.4  360.63  4782.5  359.47  4882.7  358.05  4902.8  358.37
  4922.8  357.33  4942.8  357.56  4962.9  356.78  4967.4  356.04  4970.2  355.54
  4973.4  356.04  4999.2  356.13  5057.8  358.82  5086.0  359.33  5118.3  361.50
  5227.5  365.89  5442.5  376.09  5467.9  376.93  5538.3  380.66  5538.6  380.66
#Mann=7,-1,0
  4221.2    0.05       0  4967.4    0.07       0  4973.4    0.05       0
  4999.2     0.1       0  5118.3    0.05       0  5442.5     0.1       0
  5538.3    0.05       0
Bank Sta=4967.4,4973.4
Exp/Cntr=0.3,0.1

Type RM Length L Ch R = 1,5835,472,472,472
BEGIN DESCRIPTION:
UNT 003 IN RACR 12.0
END DESCRIPTION:
XS GIS Cut Line= 3
      2207087.73     13242296.84      2207437.72     13241496.85
      2207087.72     13241096.86
#Sta/Elev= 30
  4075.2  373.08  4084.2  372.30  4097.0  372.61  4107.5  371.68  4240.9  368.98
  4293.5  367.31  4326.2  367.37  4462.3  365.34  4773.8  357.68  4811.6  356.98
  4817.4  357.61  4828.3  356.80  4872.0  356.15  4881.7  356.53  4932.4  355.25
  4955.5  354.36  4962.2  354.83  4984.0  353.91  4990.6  354.25  5001.9  353.30
  5004.6  352.80  5007.9  353.30  5012.5  354.48  5033.3  355.16  5061.8  357.36
  5096.9  356.89  5127.0  357.44  5189.0  359.22  5239.3  359.65  5479.9  368.23
#Mann=5,-1,0
  4075.2    0.05       0  4932.4     0.1       0  5001.9    0.07       0
  5007.9     0.1       0  5127.0    0.05       0
Bank Sta=5001.9,5007.9
Exp/Cntr=0.3,0.1

Type RM Length L Ch R = 1,5363,439,439,439
BEGIN DESCRIPTION:
UNT 003 IN RACR 11.0
END DESCRIPTION:
XS GIS Cut Line= 3
      2207087.74     13242446.83      2207837.72     13241646.85
      2208237.69     13241246.89
#Sta/Elev= 30
  3915.4  377.09  4035.8  373.03  4078.3  371.78  4085.1  372.05  4106.6  370.54
  4143.2  370.36  4385.5  363.28  4700.6  356.36  4792.6  355.42  4863.2  355.22
  4891.6  355.69  4898.9  354.99  4913.0  355.06  4934.1  354.04  4952.0  354.18
  4976.5  352.46  4990.7  352.32  5001.9  351.10  5004.6  350.60  5007.9  351.10
  5008.5  351.78  5026.1  352.21  5054.4  354.30  5165.1  357.20  5238.2  359.38
  5337.2  364.02  5422.1  367.25  5478.6  369.95  5563.2  374.99  5577.6  375.96
#Mann=8,-1,0
  3915.4    0.05       0  4143.2     0.1       0  4385.5    0.05       0
  4952.0     0.1       0  5001.9    0.07       0  5007.9     0.1       0
  5165.1    0.05       0  5563.2     0.1       0
Bank Sta=5001.9,5007.9
Exp/Cntr=0.3,0.1

Type RM Length L Ch R = 1,4924,442,442,442
BEGIN DESCRIPTION:
UNT 003 IN RACR 10.0
END DESCRIPTION:
XS GIS Cut Line= 3
      2207737.70     13242346.87      2208137.72     13241946.85
      2208337.71     13241546.88
#Sta/Elev= 30
  4429.1  365.74  4443.3  365.68  4556.4  361.45  4584.7  361.01  4697.8  356.85
  4712.0  355.99  4813.5  352.76  4839.2  352.47  4910.0  352.99  4922.2  352.37
  4922.3  352.36  4938.2  352.19  4966.5  351.15  4980.7  349.92  5000.2  349.59
  5002.9  349.09  5006.2  349.59  5008.8  350.10  5039.5  350.88  5061.9  352.43
  5092.6  353.22  5120.6  354.63  5142.9  354.82  5173.7  356.14  5189.8  356.36
  5330.2  361.30  5397.3  364.08  5405.7  364.83  5411.3  364.61  5442.0  365.91
#Mann=7,-1,0
  4429.1    0.05       0  4813.5     0.1       0  4922.2    0.05       0
  4922.3     0.1       0  5000.2    0.07       0  5006.2     0.1       0
  5189.8    0.05       0
Bank Sta=5000.2,5006.2
Exp/Cntr=0.3,0.1

Type RM Length L Ch R = 1,4482,488,488,488
BEGIN DESCRIPTION:
UNT 003 IN RACR 9.0
END DESCRIPTION:
XS GIS Cut Line= 3
      2207737.72     13242796.85      2208537.72     13242096.85
      2208637.72     13241696.87
#Sta/Elev= 30
  3938.1  378.77  3976.0  377.83  4086.6  374.38  4178.7  370.70  4192.9  371.05
  4221.4  369.31  4321.1  366.15  4327.7  365.35  4349.5  364.98  4370.4  363.58
  4441.6  361.79  4455.8  360.63  4540.3  357.99  4554.5  358.13  4562.1  357.29
  4583.0  357.24  4618.1  355.84  4646.6  355.84  4654.2  354.81  4752.9  353.05
  4760.5  352.30  4935.2  349.49  4991.0  347.58  4993.7  347.08  4997.0  347.58
  5049.2  349.93  5093.9  350.83  5197.0  355.66  5331.0  360.24  5413.4  364.02
#Mann=6,-1,0
  3938.1     0.1       0  3976.0    0.05       0  4935.2     0.1       0
  4991.0    0.07       0  4997.0     0.1       0  5049.2    0.05       0
Bank Sta=4991,4997
Exp/Cntr=0.3,0.1

Type RM Length L Ch R = 1,3994,414,414,414
BEGIN DESCRIPTION:
UNT 003 IN RACR 8.0
END DESCRIPTION:
XS GIS Cut Line= 3
      2208830.00     13243161.83      2208830.00     13242658.31
      2209055.69     13241842.37
#Sta/Elev= 30
  4226.1  369.84  4241.1  369.48  4291.1  365.98  4301.1  366.02  4321.1  367.64
  4331.1  367.35  4341.1  365.94  4361.1  364.72  4518.0  359.31  4727.8  351.93
  4885.7  348.56  4907.5  349.40  4917.9  348.98  4925.2  347.79  4966.1  346.69
  4990.5  346.20  4996.0  344.69  4998.8  344.19  5002.0  344.69  5004.2  345.91
  5011.3  346.48  5043.7  346.50  5249.9  353.35  5291.4  355.43  5304.7  355.44
  5312.2  356.46  5447.0  361.38  5457.6  362.41  5478.2  362.49  5576.2  367.38
#Mann=5,-1,0
  4226.1     0.1       0  4518.0    0.05       0  4966.1     0.1       0
  4996.0    0.07       0  5002.0     0.1       0
Bank Sta=4996,5002
Exp/Cntr=0.3,0.1

Type RM Length L Ch R = 1,3580,398,398,398
BEGIN DESCRIPTION:
UNT 003 IN RACR 7.0
END DESCRIPTION:
XS GIS Cut Line= 4
      2209151.20     13243048.90      2209255.35     13242771.16
      2209350.84     13242154.84      2209246.67     13241816.30
#Sta/Elev= 30
  4434.8  364.17  4618.5  356.15  4714.7  352.82  4727.3  352.08  4731.1  351.29
  4756.0  351.05  4796.5  349.20  4903.5  346.08  4976.6  344.16  4979.4  343.66
  4982.6  344.16  4988.8  344.97  4998.9  344.27  5042.6  344.86  5120.3  347.06
  5150.7  348.55  5231.6  350.46  5236.7  351.47  5241.8  351.01  5322.7  354.03
  5373.9  355.13  5394.8  356.36  5426.2  357.08  5436.7  358.25  5451.5  358.07
  5457.6  358.96  5549.6  361.67  5645.9  366.71  5685.6  366.94  5709.3  367.87
#Mann=4,-1,0
  4434.8    0.05       0  4903.5     0.1       0  4976.6    0.07       0
  4982.6     0.1       0
Bank Sta=4976.6,4982.6
Exp/Cntr=0.3,0.1

Type RM Length L Ch R = 1,3182,262,262,262
BEGIN DESCRIPTION:
UNT 003 IN RACR 6.0
END DESCRIPTION:
XS GIS Cut Line= 3
      2209387.74     13243096.82      2209637.72     13242696.85
      2210137.74     13241896.82
#Sta/Elev= 30
  4513.6  362.02  4521.2  361.17  4536.6  361.18  4548.9  359.80  4615.6  356.79
  4643.3  356.36  4652.1  355.47  4752.4  351.84  4840.8  347.83  4929.2  345.21
  4988.2  343.18  4989.9  342.24  4992.7  341.74  4995.9  342.24  5008.3  342.88
  5050.7  342.61  5102.6  343.92  5275.9  345.69  5406.8  349.65  5412.7  350.56
  5428.1  349.89  5565.7  355.52  5610.3  356.45  5616.7  356.78  5622.6  358.42
  5632.1  357.73  5645.6  358.54  5681.0  358.50  5699.8  359.68  5928.7  367.19
#Mann=6,-1,0
  4513.6    0.05       0  4929.2     0.1       0  4989.9    0.07       0
  4995.9     0.1       0  5565.7    0.08       0  5699.8     0.1       0
Bank Sta=4989.9,4995.9
Exp/Cntr=0.3,0.1

Type RM Length L Ch R = 1,2920,87,87,87
BEGIN DESCRIPTION:
Mapping XS 50048ca4
END DESCRIPTION:
XS GIS Cut Line= 2
      2209563.23     13243227.50      2210410.49     13241932.30
#Sta/Elev= 30
  4394.0  362.96  4503.1  357.76  4508.9  357.50  4691.0  349.75  4740.4  348.07
  4860.7  345.30  4878.9  345.29  4896.6  345.48  4909.6  342.32  4924.7  340.36
  4932.5  337.58  4945.8  335.70  4971.9  335.00  4988.1  334.81  4990.8  334.31
  4994.1  334.81  5027.3  335.11  5066.9  337.14  5120.7  342.80  5203.4  344.27
  5254.8  347.06  5319.2  348.74  5401.1  351.36  5410.3  352.49  5442.7  352.82
  5488.6  354.76  5553.9  355.59  5569.9  356.87  5757.0  362.87  5941.7  366.71
#Mann=16,-1,0
  4394.0    0.05       0  4503.1    0.08       0  4508.9    0.05       0
  4691.0    0.08       0  4740.4    0.05       0  4860.7     0.1       0
  4878.9    0.08       0  4971.9     0.1       0  4988.1    0.07       0
  4994.1     0.1       0  5066.9    0.08       0  5203.4     0.1       0
  5254.8    0.08       0  5319.2     0.1       0  5442.7    0.08       0
  5569.9     0.1       0
Bank Sta=4988.1,4994.1
Exp/Cntr=0.3,0.1

Type RM Length L Ch R = 1,2833,106,106,106
BEGIN DESCRIPTION:
Mapping XS 3e90d057
END DESCRIPTION:
XS GIS Cut Line= 2
      2209618.78     13243293.48      2210472.85     13241974.19
#Sta/Elev= 30
  4404.4  364.05  4592.7  355.48  4594.1  355.40  4662.5  353.30  4668.8  352.29
  4684.0  352.70  4741.4  350.49  4782.1  350.38  4824.9  350.10  4928.7  350.55
  4971.6  349.61  5055.8  347.92  5079.7  348.19  5088.9  347.81  5094.9  346.35
  5125.2  346.51  5131.1  344.57  5146.3  345.74  5152.3  344.33  5161.0  344.24
  5164.4  342.72  5167.2  342.22  5170.4  342.72  5286.6  346.08  5318.5  347.81
  5350.4  348.10  5424.7  350.45  5499.8  351.89  5682.6  357.81  5976.0  365.11
#Mann=14,-1,0
  4404.4    0.08       0  4592.7    0.05       0  4594.1    0.08       0
  4782.1    0.05       0  4824.9    0.08       0  4971.6    0.05       0
  5055.8    0.08       0  5161.0    0.05       0  5164.4    0.03       0
  5170.4    0.05       0  5286.6    0.08       0  5350.4     0.1       0
  5424.7    0.08       0  5682.6     0.1       0
Bank Sta=5164.4,5170.4
Exp/Cntr=0.3,0.1

Type RM Length L Ch R = 1,2727,488,488,488
BEGIN DESCRIPTION:
UNT 003 IN RACR 5.0
END DESCRIPTION:
XS GIS Cut Line= 2
      2209674.37     13243335.09      2210608.39     13242022.61
#Sta/Elev= 30
  4398.7  364.10  4404.3  363.89  4472.1  360.29  4641.7  353.02  4648.9  352.64
  4808.7  346.35  4966.1  343.21  5022.7  344.10  5031.3  345.84  5046.1  346.98
  5052.2  346.54  5059.3  349.24  5067.0  349.38  5087.9  348.62  5102.6  343.02
  5117.4  341.03  5142.2  340.24  5145.0  339.74  5148.2  340.24  5353.9  347.20
  5417.4  347.74  5446.9  349.45  5533.0  351.43  5539.1  350.83  5621.3  353.70
  5801.0  358.09  5898.2  360.50  5913.0  361.92  5933.9  361.63  6009.6  363.76
#Mann=9,-1,0
  4398.7    0.05       0  4404.3    0.08       0  4472.1    0.05       0
  4641.7    0.08       0  4648.9    0.05       0  5142.2    0.03       0
  5148.2    0.05       0  5621.3    0.08       0  5801.0     0.1       0
Bank Sta=5142.2,5148.2
Exp/Cntr=0.3,0.1

Type RM Length L Ch R = 1,2239,462,462,462
BEGIN DESCRIPTION:
UNT 003 IN RACR 4.0
END DESCRIPTION:
XS GIS Cut Line= 3
      2209737.73     13243746.84      2210487.72     13242946.85
      2210987.74     13242146.83
#Sta/Elev= 30
  3879.5  376.75  4067.3  367.60  4120.1  364.20  4141.1  366.02  4183.6  362.38
  4579.7  346.58  4728.7  342.11  4912.7  338.96  4986.6  337.58  4989.4  337.08
  4992.6  337.58  5047.4  338.40  5062.7  342.18  5070.4  342.40  5099.3  342.61
  5120.5  340.27  5141.8  341.28  5151.2  344.28  5164.8  345.53  5178.3  345.16
  5187.7  341.79  5193.6  342.14  5209.0  339.65  5251.4  340.01  5266.8  342.97
  5272.7  342.30  5282.1  343.95  5592.2  353.88  5875.7  366.50  5919.5  368.18
#Mann=6,-1,0
  3879.5     0.1       0  4067.3    0.05       0  4912.7     0.1       0
  4986.6    0.07       0  4992.6     0.1       0  5875.7    0.08       0
Bank Sta=4986.6,4992.6
Exp/Cntr=0.3,0.1

Type RM Length L Ch R = 1,1777,461,461,461
BEGIN DESCRIPTION:
UNT 003 IN RACR 3.0
END DESCRIPTION:
XS GIS Cut Line= 3
      2210437.75     13243646.82      2210837.72     13243246.85
      2211187.74     13242446.81
#Sta/Elev= 30
  4410.4  352.35  4687.5  342.24  4721.5  340.35  4749.8  340.98  4763.9  342.78
  4792.2  339.39  4908.5  337.67  4961.9  337.46  4997.9  336.53  5063.1  336.51
  5065.8  336.01  5069.1  336.51  5091.7  336.78  5250.0  337.98  5392.0  340.51
  5415.4  342.52  5423.6  345.85  5433.3  346.76  5438.8  346.70  5456.3  343.87
  5462.2  341.28  5491.0  339.48  5500.0  341.16  5514.4  342.29  5521.8  345.25
  5538.0  346.01  5652.8  350.86  5689.0  351.81  5696.4  352.85  5849.3  358.46
#Mann=8,-1,0
  4410.4    0.05       0  4687.5     0.1       0  4908.5    0.05       0
  5063.1    0.03       0  5069.1    0.05       0  5091.7     0.1       0
  5250.0    0.05       0  5538.0     0.1       0
Bank Sta=5063.1,5069.1
Exp/Cntr=0.3,0.1

Type RM Length L Ch R = 1,1316,482,482,482
BEGIN DESCRIPTION:
UNT 003 IN RACR 2.0
END DESCRIPTION:
XS GIS Cut Line= 3
      2210487.73     13244096.84      2211287.72     13243346.85
      2211237.72     13242546.88
#Sta/Elev= 30
  3915.7  360.69  4071.3  353.94  4156.2  348.55  4312.1  347.75  4333.1  345.79
  4340.4  343.30  4361.4  341.85  4410.7  340.84  4446.4  341.88  4474.7  338.42
  4565.4  336.61  4638.9  335.75  4863.5  336.19  4973.9  334.50  4976.6  334.00
  4979.9  334.50  5012.7  334.54  5178.1  335.37  5322.9  336.67  5433.1  339.31
  5493.2  341.76  5553.3  347.51  5563.3  347.34  5593.4  341.44  5613.4  340.69
  5643.5  344.51  5653.5  347.38  5673.6  349.30  5773.2  353.68  5813.8  354.84
#Mann=8,-1,0
  3915.7    0.05       0  4565.4     0.1       0  4638.9    0.05       0
  4973.9    0.03       0  4979.9    0.05       0  5012.7     0.1       0
  5178.1    0.05       0  5773.2     0.1       0
Bank Sta=4973.9,4979.9
Exp/Cntr=0.3,0.1
