--- UNT 005 IN RACR.prj (project) ---

Proj Title=UNT 005 IN RACR Base Level Engineering
Current Plan=p01
Default Exp/Contr=0.3,0.1
English Units
Geom File=g01
Flow File=f01
Plan File=p01
Y Axis Title=Elevation
X Axis Title(PF)=Main Channel Distance
X Axis Title(XS)=Station
BEGIN DESCRIPTION:
UNT 005 IN RACR
END DESCRIPTION:
DSS Export Rating Curves= 0
DSS Export Rating Curve Sorted= 0
DSS Export Volume Flow Curves= 0
DXF OffsetX= 0
DXF OffsetY= 0
DXF ScaleX= 1
DXF ScaleY= 10

--- UNT 005 IN RACR.p01 (plan) ---

Plan Title=Multiple Run
Short Identifier=Multiple
Geom File=g01
Flow File=f01
Subcritical Flow
K Sum by GR= 0
Std Step Tol= 0.01
Critical Tol= 0.01
Num of Std Step Trials= 20
Max Error Tol= 0.3
Flow Tol Ratio= 0.001
Split Flow NTrial= 30
Split Flow Tol= 0.02
Split Flow Ratio= 0.02
Log Output Level= 0
Friction Slope Method= 1
Unsteady Friction Slope Method= 2
Unsteady Bridges Friction Slope Method= 1
Parabolic Critical Depth
Global Vel Dist=  1 , 1 , 1
Global Log Level= 0
CheckData=True
Encroach Param= -1, 0, 0, 0
BEGIN DESCRIPTION:
Multiple Run
END DESCRIPTION:

--- UNT 005 IN RACR.f01 (steady flow) ---

Flow Title=Multiple
Program Version=4.10
Number of Profiles= 7
Profile Names=10-year,25-year,50-year,1pct_min,100-year,1pct_plu,500-year
River Rch & RM=UNT 005 IN RACR,Reach-1         ,17754
     193     267     328     297     402     543     612
River Rch & RM=UNT 005 IN RACR,Reach-1         ,17393
     242     337     417     379     512     693     787
River Rch & RM=UNT 005 IN RACR,Reach-1         ,13224
     332     469     585     537     726     982    1134
River Rch & RM=UNT 005 IN RACR,Reach-1         ,8285
     420     600     753     694     938    1269    1481
Boundary for River Rch & Prof#=UNT 005 IN RACR,Reach-1         , 1
Up Type= 0
Dn Type= 3
Dn Slope=0.005
Boundary for River Rch & Prof#=UNT 005 IN RACR,Reach-1         , 2
Up Type= 0
Dn Type= 3
Dn Slope=0.005
Boundary for River Rch & Prof#=UNT 005 IN RACR,Reach-1         , 3
Up Type= 0
Dn Type= 3
Dn Slope=0.005
Boundary for River Rch & Prof#=UNT 005 IN RACR,Reach-1         , 4
Up Type= 0
Dn Type= 3
Dn Slope=0.005
Boundary for River Rch & Prof#=UNT 005 IN RACR,Reach-1         , 5
Up Type= 0
Dn Type= 3
Dn Slope=0.005
Boundary for River Rch & Prof#=UNT 005 IN RACR,Reach-1         , 6
Up Type= 0
Dn Type= 3
Dn Slope=0.005
Boundary for River Rch & Prof#=UNT 005 IN RACR,Reach-1         , 7
Up Type= 0
Dn Type= 3
Dn Slope=0.005
DSS Import GetInterval= 0
DSS Import GetPeak= 0
DSS Import FillOption= 0

--- UNT 005 IN RACR.g01 (geometry) ---

Geom Title=Existing Conditions
Program Version=4.10

River Reach=UNT 005 IN RACR ,Reach-1
Reach XY= 30
      2201763.73     13236766.09       2202804.3     13236237.26
      2203467.67     13235724.21      2203904.86      13235845.7
      2203915.28     13236322.09      2204122.84     13236504.08
      2204281.94     13236927.65      2204548.45     13237105.05
      2205219.72     13237244.45      2205884.43      13237742.7
      2206570.61      13237821.2      2207139.24      13238183.2
       2207992.6      13238246.5      2209234.57     13237661.84
      2210406.23     13237424.11       2210624.5     13237225.52
      2210870.06      13236598.3      2211033.63      13236575.5
      2211108.12     13236186.91      2211897.86     13235836.32
       2211890.7     13235508.01      2212214.82     13235241.08
      2212578.63     13235444.32      2213003.18     13235297.66
      2213581.94     13235348.69      2214315.24     13235831.27
      2214774.74     13235917.61      2214949.91     13235442.19
      2215180.64     13235423.96      2215372.23     13235230.33

Type RM Length L Ch R = 1 ,17754   ,361,361,361
BEGIN DESCRIPTION:
UNT 005 IN RACR 36.0
END DESCRIPTION:
XS GIS Cut Line= 3
      2201887.72     13237196.81      2201887.72     13236646.85
      2201987.71     13236046.89
#Sta/Elev= 30
    4478  397.76    4548  396.03    4648  391.86    4748  389.13    4858  385.35
    4968  382.82    4988  381.31  5007.7  379.73  5025.5  380.94  5038.1   381.1
  5055.8  382.33  5088.8  382.23  5129.3  380.76  5139.5  382.07  5159.8  382.33
  5169.9   382.3  5182.6     381  5190.2  381.78  5220.6  382.75    5251  382.58
  5281.4  383.49  5332.1  384.09  5433.5  387.05  5499.6  390.07  5585.5  393.38
    5596  394.36  5599.2  394.27  5608.4  394.03    5616  394.83  5636.2  395.57
#Mann= 5 ,-1 , 0
    4478     .05       0    4988     .05       0  5499.6      .1       0
    5596     .05       0  5599.2      .1       0
Bank Sta=4988,5038.1
XS Rating Curve= 0 ,0
Exp/Cntr=0.3,0.1

Type RM Length L Ch R = 1 ,17393   ,116,116,116
BEGIN DESCRIPTION:
Mapping XS 3e9bf1e3
END DESCRIPTION:
XS GIS Cut Line= 4
      2202056.54     13237148.42      2202223.39     13236665.44
      2202176.56      13236366.9      2202018.49     13236062.47
#Sta/Elev= 30
  4315.2  393.32  4412.1  391.85    4427  390.93    4640  386.65  4830.2  381.95
  4855.1  381.78  4875.4  383.48  4885.5  386.45  4892.8  387.04  4897.8  386.86
  4908.4  384.54  4915.9  383.85    4926  380.39  4936.1     378  4946.2  377.01
  5028.2  376.79  5047.2  375.97  5085.7   378.4  5090.8  379.56  5098.1  382.51
  5125.9  386.92    5141  386.06    5151  384.75  5157.5  382.99    5196  383.41
    5220  384.46  5387.6  390.72  5417.3  392.96  5446.2  393.61  5471.4  394.64
#Mann= 6 ,-1 , 0
  4315.2     .05       0  4908.4     .07       0    4926     .05       0
  5090.8      .1       0    5220     .05       0  5446.2      .1       0
Bank Sta=4926,5090.8
XS Rating Curve= 0 ,0
Exp/Cntr=0.3,0.1

Type RM Length L Ch R = 1 ,17277   ,59,59,59
BEGIN DESCRIPTION:
Mapping XS 2a5477c3
END DESCRIPTION:
XS GIS Cut Line= 4
      2202405.21      13237234.1      2202349.65       13236557.
      2202287.15     13236411.17      2202027.76     13236020.35
#Sta/Elev= 30
  4200.7  389.79  4298.3  386.68  4428.7  386.24  4479.8  385.02  4569.2  384.69
  4601.1  383.42  4649.4  383.61  4722.5  382.16  4848.4  380.94  4882.9  381.47
  4912.9  383.79  4926.1  383.04  4934.6  380.21  4956.4  377.16  4978.7  376.13
  4996.8   376.2    5002  375.48  5010.8  376.41  5069.4  377.06  5078.4  378.13
  5084.4  378.13  5099.5  380.78  5114.5  382.57  5127.9  385.25  5150.6   382.7
  5186.9   383.2    5308  388.42  5373.1  390.24  5428.9  393.03  5507.8  395.71
#Mann= 6 ,-1 , 0
  4200.7     .05       0  4848.4      .1       0  4934.6     .05       0
  5099.5      .1       0  5186.9     .05       0  5428.9      .1       0
Bank Sta=4934.6,5099.5
XS Rating Curve= 0 ,0
Exp/Cntr=0.3,0.1

Type RM Length L Ch R = 1 ,17218   ,73,73,73
BEGIN DESCRIPTION:
Mapping XS 2e1fc7ad
END DESCRIPTION:
XS GIS Cut Line= 4
      2202432.99     13237209.82      2202384.37     13236487.56
      2202332.29      13236369.5      2202054.53     13236008.41
#Sta/Elev= 30
  4205.6  389.68  4258.7  388.08  4338.9  388.01  4714.4  382.53  4827.1  380.95
    4860   380.6  4870.1  381.98  4900.1  383.68  4952.1   384.8    4958   383.9
  4963.4  381.47    4974  379.43    4982  381.12  4986.8  381.29  4995.8  378.07
  5004.4  377.28  5007.6  377.78  5010.1   379.5  5017.7  379.47  5030.7  381.43
  5033.4  381.96  5039.6  384.11  5050.5   385.3  5085.7   385.5  5106.5  383.45
  5112.8   385.6    5121  382.66  5159.2  381.99  5471.4  393.69  5514.1  395.01
#Mann= 7 ,-1 , 0
  4205.6     .05       0  4714.4      .1       0  4827.1     .05       0
  5033.4     .07       0  5039.6      .1       0  5159.2     .05       0
  5471.4      .1       0
Bank Sta=4982,5030.7
XS Rating Curve= 0 ,0
Exp/Cntr=0.3,0.1

Type RM Length L Ch R = 1 ,17145   ,257,257,257
BEGIN DESCRIPTION:
UNT 005 IN RACR 35.0
END DESCRIPTION:
XS GIS Cut Line= 4
      2202464.24     13237216.76       2202443.4     13236435.48
      2202394.79     13236341.73      2202092.72     13236008.41
#Sta/Elev= 30
  4176.6  390.31  4256.5  389.42  4276.5  388.77  4356.6  388.19  4426.6  386.89
  4496.6  386.34  4536.6  385.32  4605.1  384.45  4616.7  383.83  4781.4  381.38
  4802.1  380.94  4826.7  380.93  4886.8  379.78  4967.9  379.49  4983.1  379.01
  4990.4  379.29  5002.2  378.87  5004.9  378.37  5012.9   379.3  5021.7  379.41
    5072  379.08  5114.5   379.7  5130.7  380.22  5256.5  384.34  5362.6  388.91
  5433.6  391.13  5440.3  391.68  5468.7  392.24  5475.4  393.08  5513.6  394.21
#Mann= 6 ,-1 , 0
  4176.6     .05       0  4781.4      .1       0  4802.1     .05       0
  4886.8     .03       0  5114.5      .1       0  5130.7     .05       0
Bank Sta=4886.8,5114.5
XS Rating Curve= 0 ,0
Exp/Cntr=0.3,0.1

Type RM Length L Ch R = 1 ,16888   ,359,359,359
BEGIN DESCRIPTION:
UNT 005 IN RACR 34.0
END DESCRIPTION:
XS GIS Cut Line= 4
       2202865.2      13236916.8      2202764.13     13236478.83
      2202460.91     13235993.68      2202225.23     13235791.67
#Sta/Elev= 30
  4318.5  400.18  4369.3  398.21    4380  397.32  4431.3   395.6  4555.8  389.56
    4684  384.43  4825.3  379.58  4904.3  378.33  4962.1   377.4  4970.8  377.87
  4992.8  377.69  4998.7  377.22  5006.2  377.65  5050.5  377.38  5064.9   376.4
  5077.7  377.47  5108.3  378.28  5114.2  378.42  5346.9  383.83  5361.2  384.76
  5375.4  384.76    5404  386.12  5481.9  388.37  5567.5  391.58  5595.2  392.01
  5602.6  391.84  5623.5   393.1  5631.2  392.76  5646.2  393.25  5650.5   393.5
#Mann= 5 ,-1 , 0
  4318.5     .05       0  4904.3     .03       0  5108.3     .05       0
  5595.2      .1       0  5646.2     .05       0
Bank Sta=4904.3,5114.2
XS Rating Curve= 0 ,0
Exp/Cntr=0.3,0.1

Type RM Length L Ch R = 1 ,16529   ,513,513,513
BEGIN DESCRIPTION:
UNT 005 IN RACR 33.0
END DESCRIPTION:
XS GIS Cut Line= 4
      2202979.75     13236795.47      2203047.13     13236303.64
       2202811.3     13235852.18       2202443.4     13235631.45
#Sta/Elev= 30
  4308.6   396.4  4475.8  389.16  4488.9   389.1    4499  388.36  4630.2  384.26
  4650.4  383.23  4761.4  380.47  4781.6   380.4  4891.7   377.4  4899.1  377.66
  4936.8  376.72  4981.8  375.91  5038.3  376.18  5047.8  375.28  5053.7  376.04
  5075.8  375.81  5097.8  376.26    5106  375.91  5151.1  376.86  5218.8  377.98
  5246.8  378.77  5252.7  379.34  5297.8  379.78  5372.2  382.01  5387.7  382.11
  5393.5  382.65  5568.5  388.03  5642.3  389.93  5727.9  391.23  5743.4  391.82
#Mann= 3 , 0 , 0
  4308.6     .05       0  4936.8     .03       0  5151.1     .05       0
Bank Sta=4936.8,5151.1
XS Rating Curve= 0 ,0
Exp/Cntr=0.3,0.1

Type RM Length L Ch R = 1 ,16016   ,435,435,435
BEGIN DESCRIPTION:
UNT 005 IN RACR 32.0
END DESCRIPTION:
XS GIS Cut Line= 4
      2203242.52     13236472.11      2203451.41      13236067.8
      2203040.39      13235164.9      2202919.12     13234996.46
#Sta/Elev= 30
  4269.8  383.76  4314.5  382.83  4353.1   383.1  4380.9   382.5  4419.6  382.59
  4425.2  382.08  4441.7  382.54  4469.5  381.91  4530.3  381.92  4613.3  381.16
  4701.9  379.56  4707.5  379.98  4744.1   379.5  4893.5  375.31  4901.7  375.19
  4916.5  374.53  4985.7  373.97  5000.4  372.98  5022.6  374.31    5135   374.3
  5204.2  375.31  5491.5  379.44  5589.5  379.92  5658.7   381.2  5714.1  383.29
  5739.2  383.27  5752.4  384.36  5767.1   384.2  5845.5  386.62  5924.5   389.2
#Mann= 5 ,-1 , 0
  4269.8     .05       0  4893.5     .07       0  5204.2     .05       0
  5491.5      .1       0  5845.5     .05       0
Bank Sta=4901.7,5204.2
XS Rating Curve= 0 ,0
Exp/Cntr=0.3,0.1

Type RM Length L Ch R = 1 ,15581   ,131,131,131
BEGIN DESCRIPTION:
Mapping XS a043ac0d
END DESCRIPTION:
XS GIS Cut Line= 5
       2203115.3     13236938.92      2203501.56     13236483.22
      2203675.17     13236162.04      2203696.87     13235697.63
      2203770.66     13235011.88
#Sta/Elev= 30
  3724.2  398.95  4138.8  381.58  4294.8  376.71  4411.1  374.43  4634.8  373.37
  4640.4  372.38  4678.5  372.65  4688.9  371.93    4842  374.22  4962.2  373.06
  4992.2  372.19  5102.3     373  5192.6  373.09    5253  375.36  5273.1  376.23
  5307.1  375.84  5406.1  375.03  5474.2  375.28    5483  376.22    5488  375.59
  5594.9  378.53  5625.1  380.37  5655.3   380.3  5665.3  380.81    5672  382.25
  5705.5  382.45    5764  385.22    5769  384.45  5796.1  387.39  5841.3  387.48
#Mann= 5 ,-1 , 0
  3724.2     .08       0  4962.2     .07       0    5253     .08       0
  5307.1     .05       0  5406.1      .1       0
Bank Sta=4962.2,5102.3
XS Rating Curve= 0 ,0
Exp/Cntr=0.3,0.1

Type RM Length L Ch R = 1 ,15450   ,698,698,698
BEGIN DESCRIPTION:
Mapping XS 2bee923e
END DESCRIPTION:
XS GIS Cut Line= 4
      2203123.99     13237017.04      2203614.41     13236509.26
       2203753.3      13236157.7      2203905.21     13235063.95
#Sta/Elev= 30
  3581.3  402.88  3591.2  401.53  3598.1  402.15  3640.6  400.59  3647.8  399.36
  3697.2  397.79  3704.4  396.56  3739.6   395.6  3746.8  394.43  3796.2  393.22
  3803.4  391.82  3824.5  392.04  3831.7  390.45  3895.3  387.09  3951.9  384.64
  3958.8  385.38    3966  383.76    4072  379.24  4262.9  372.72  4475.6  370.57
  4989.2  372.59  4999.3  371.65  5049.7  372.19  5069.9  371.28  5101.2  372.64
  5150.7  373.92    5181   372.6  5403.1   374.3  5536.4   377.4  5769.5  386.57
#Mann= 3 , 0 , 0
  3581.3     .08       0  4989.2     .07       0  5101.2     .08       0
Bank Sta=4989.2,5101.2
XS Rating Curve= 0 ,0
Exp/Cntr=0.3,0.1

Type RM Length L Ch R = 1 ,14752   ,280,280,280
BEGIN DESCRIPTION:
UNT 005 IN RACR 31.0
END DESCRIPTION:
XS GIS Cut Line= 4
      2203363.82     13237091.99       2203801.8     13236627.06
      2204307.15     13235899.35      2204617.06     13235778.08
#Sta/Elev= 30
  4059.5  398.82    4094  396.38  4221.4  391.34  4234.3  389.53  4470.4  377.44
    4554   374.1  4589.2  373.99    4738  368.83    4896  368.48  4990.7  367.65
  4997.1   366.5  5018.3  367.99  5054.1  367.11  5089.9  368.36  5112.4  367.94
  5170.2  369.89  5220.9  368.64  5283.7  369.49  5288.1  369.48  5349.2  368.82
    5385  372.07  5420.8  373.56  5528.2  377.57    5617  379.58  5662.5  381.49
    5687  383.55  5810.3  387.76  5825.4  387.35  5831.8  388.59    5917  391.63
#Mann= 7 ,-1 , 0
  4059.5      .1       0  4234.3     .05       0  4470.4      .1       0
    4896     .07       0  5089.9      .1       0  5283.7     .08       0
  5288.1      .1       0
Bank Sta=4896,5089.9
XS Rating Curve= 0 ,0
Exp/Cntr=0.3,0.1

Type RM Length L Ch R = 1 ,14472   ,197,197,197
BEGIN DESCRIPTION:
UNT 005 IN RACR 30.0
END DESCRIPTION:
XS GIS Cut Line= 3
      2203337.73     13237396.85      2204137.72     13236596.85
      2204537.75     13236246.83
#Sta/Elev= 30
  3843.4  409.09  3857.5  409.15  3915.5  405.51  3984.8  402.56    3999  401.11
  4055.5  398.78  4083.8  396.44  4112.1  395.73  4154.5  392.88  4225.2  390.21
  4267.8  386.93  4366.6  383.25    4413  380.47  4437.4  379.93  4479.8  376.82
  4508.1  377.08  4536.4  374.08  4635.3  371.56  4720.2  367.89  4960.6  365.69
  4981.9  366.86  5010.1  362.57  5024.6  365.88  5045.5  366.66  5052.6  366.41
  5091.9  367.18  5300.8  373.02  5343.5   375.6  5392.8  376.34  5506.3  381.28
#Mann= 8 ,-1 , 0
  3843.4     .08       0  3915.5      .1       0  4267.8     .05       0
    4413      .1       0  4981.9     .07       0  5045.5      .1       0
  5052.6     .08       0  5091.9      .1       0
Bank Sta=4981.9,5045.5
XS Rating Curve= 0 ,0
Exp/Cntr=0.3,0.1

Type RM Length L Ch R = 1 ,14275   ,60,60,60
BEGIN DESCRIPTION:
Mapping XS 0b3c79e9
END DESCRIPTION:
XS GIS Cut Line= 6
      2203472.03     13237282.71      2204048.44     13236775.75
      2204149.13     13236793.12      2204242.88     13236751.45
      2204232.46       13236682.      2204652.59     13236327.85
#Sta/Elev= 30
    4066  400.23  4138.3  395.81  4159.1  395.84  4279.6   389.4  4317.5   386.6
  4428.6   382.3  4442.8  380.67  4485.5  379.49  4525.5  376.76  4790.1  366.59
  4835.8  366.18  4863.3  368.68    4869  367.86    4874  369.77  4893.8  365.74
  4923.8  360.27  4945.2  358.69  5032.1  357.13  5043.8  358.27  5083.5  366.19
  5107.8  366.21  5123.2  367.88  5129.7  366.25    5144  366.11  5151.8  364.53
  5163.3  366.39  5224.9  368.09  5258.4  367.81  5314.4  370.69  5658.1  383.03
#Mann= 7 ,-1 , 0
    4066      .1       0  4317.5     .05       0  4525.5      .1       0
  4893.8     .07       0  5083.5      .1       0  5163.3     .08       0
  5224.9      .1       0
Bank Sta=4893.8,5083.5
XS Rating Curve= 0 ,0
Exp/Cntr=0.3,0.1

Type RM Length L Ch R = 1 ,14215   ,90,90,90
BEGIN DESCRIPTION:
Mapping XS eca22372
END DESCRIPTION:
XS GIS Cut Line= 6
      2203468.56     13237313.96      2204083.16     13236810.48
      2204138.71      13236869.5      2204308.85     13236779.23
      2204288.02     13236713.25       2204735.9     13236334.81
#Sta/Elev= 30
  4025.2  401.56    4037  401.76  4128.6  395.49  4165.2  394.61  4206.8   391.4
  4256.8  389.76  4304.5  386.08  4577.5  374.03  4789.6  365.43    4804  367.22
  4818.3  371.52  4916.8  370.95  4967.6  367.87  4977.1  368.88  5012.8   367.7
  5070.8  368.96  5080.8  370.56  5112.7  369.92  5117.9  367.03  5127.3  367.17
  5137.8   369.7  5150.2  369.16  5162.5  370.37  5195.3  363.96  5201.8  366.24
  5221.2  366.61  5283.5  368.28  5634.8  380.95  5649.1  382.38  5748.9  384.96
#Mann= 7 ,-1 , 0
  4025.2      .1       0  4304.5     .05       0  4577.5      .1       0
  4916.8     .07       0  5070.8      .1       0  5221.2     .08       0
  5283.5      .1       0
#XS Ineff= 2 , 0
         4875.89  371.94 5158.75          370.34
Permanent Ineff=
       F       F
Bank Sta=4916.8,5080.8
XS Rating Curve= 0 ,0
Exp/Cntr=0.3,0.1

Type RM Length L Ch R = 1 ,14125   ,313,313,313
BEGIN DESCRIPTION:
Mapping XS a417ee6c
END DESCRIPTION:
XS GIS Cut Line= 3
      2203461.61     13237352.16       2204378.3     13236841.73
      2204773.42       13236457.
#Sta/Elev= 30
  4076.2   403.4  4106.1  400.92  4142.3  399.96  4266.9  392.53  4277.2  392.85
    4335  389.78  4405.2  384.91  4553.9  377.99  4563.9  376.83  4598.3  376.93
  4629.3  374.13  4659.5  374.02  4672.8  372.62  4724.2  371.22  4781.4  368.15
  4894.6  365.88  4900.3  365.61  4997.5  364.31  5084.4  365.35  5106.1  364.58
  5113.1  363.23  5122.1  364.83  5163.9  365.65  5182.8  365.86  5255.7  367.82
    5284  367.45  5298.2  368.85    5390  371.68  5491.4  376.27  5676.9  383.07
#Mann= 7 ,-1 , 0
  4076.2      .1       0  4405.2     .05       0  4659.5      .1       0
  4894.6     .07       0  5163.9      .1       0  5182.8     .08       0
  5491.4      .1       0
Bank Sta=4900.3,5163.9
XS Rating Curve= 0 ,0
Exp/Cntr=0.3,0.1

Type RM Length L Ch R = 1 ,13812   ,305,305,305
BEGIN DESCRIPTION:
Mapping XS 0c29d7e5
END DESCRIPTION:
XS GIS Cut Line= 3
      2204350.37     13237739.37      2204541.35     13236949.41
      2204783.56     13236499.59
#Sta/Elev= 30
  4320.6  385.02  4376.5  383.85  4405.5  381.56  4460.2  380.66  4467.2  379.28
  4487.8  377.69  4518.7  376.92    4546  375.21  4590.9  374.18  4627.6  372.06
  4674.6   371.6  4683.3  370.07  4734.7  367.89    4745  368.37  4775.9  366.71
  4800.1  366.77  4847.9  364.75  4868.5  365.35  4919.9  364.11  4991.7  362.11
  5009.4  362.86  5147.6  364.05  5204.8   365.9  5241.7  365.82  5302.9  369.12
  5390.5  371.97    5451  374.93  5560.6  378.71  5625.8   381.2  5644.2  382.59
#Mann= 7 ,-1 , 0
  4320.6     .05       0    4546      .1       0  4919.9     .07       0
  5147.6     .08       0  5241.7      .1       0    5451     .08       0
  5560.6      .1       0
Bank Sta=4919.9,5147.6
XS Rating Curve= 0 ,0
Exp/Cntr=0.3,0.1

Type RM Length L Ch R = 1 ,13507   ,283,283,283
BEGIN DESCRIPTION:
Mapping XS f0cd0fcc
END DESCRIPTION:
XS GIS Cut Line= 4
      2204953.67     13237769.74      2205105.59     13237457.22
      2204688.92     13237023.19      2204819.13     13236524.04
#Sta/Elev= 30
  4209.5  377.83  4229.8     378  4235.4  376.56  4297.5  372.59    4335   371.4
  4357.3  369.56  4393.2  368.81  4432.8  365.96  4485.4  363.82  4535.2   362.1
  4647.7  361.44  4796.1   362.4  4803.3  361.61  4810.3  362.99  4824.4  363.31
  4838.6  361.87  4944.9   362.1  4951.8  362.47    4987   360.7  4994.2  361.71
  5029.5  362.45  5101.9  362.59  5140.9   363.4  5215.3  364.21  5369.3  369.37
  5423.6  371.59  5450.2  373.72  5614.9   379.4  5632.2  380.37  5674.5  381.55
#Mann= 9 ,-1 , 0
  4209.5      .1       0  4485.4     .08       0  4944.9     .07       0
  5029.5     .08       0  5101.9      .1       0  5140.9     .08       0
  5215.3      .1       0  5614.9     .08       0  5632.2      .1       0
Bank Sta=4951.8,5029.5
XS Rating Curve= 0 ,0
Exp/Cntr=0.3,0.1

Type RM Length L Ch R = 1 ,13224   ,460,460,460
BEGIN DESCRIPTION:
Mapping XS 47368637
END DESCRIPTION:
XS GIS Cut Line= 4
      2205079.57     13237808.75      2205261.84     13237483.26
      2204892.91     13237070.94      2205001.06     13236499.91
#Sta/Elev= 30
  4308.1  375.46  4390.5  371.28  4402.1  369.76  4455.7  368.29  4497.4  365.89
  4564.2  363.16  4596.1  363.13  4608.3  361.66  4617.8  361.73  4639.5  360.49
  4661.2  360.71  4688.7  359.64  4695.6  360.35  5014.1  361.04  5042.5  361.87
    5050  361.64  5098.6     362  5141.1   362.3  5226.5  362.93  5370.9  366.97
  5482.8  370.57  5533.7  373.16  5594.8  374.83  5676.2  378.02  5686.4  379.02
  5714.4   379.1  5719.5  379.72  5727.1  379.25  5768.3  381.55  5815.6  383.49
#Mann= 7 ,-1 , 0
  4308.1      .1       0  4497.4     .08       0  4617.8     .07       0
    5050      .1       0  5098.6     .08       0  5141.1      .1       0
  5768.3     .08       0
Bank Sta=4617.8,5042.5
XS Rating Curve= 0 ,0
Exp/Cntr=0.3,0.1

Type RM Length L Ch R = 1 ,12764   ,194,194,194
BEGIN DESCRIPTION:
Mapping XS ba60787c
END DESCRIPTION:
XS GIS Cut Line= 4
      2205070.83     13237878.26      2205326.94     13237613.47
      2205522.25     13237101.32      2206038.62     13236671.74
#Sta/Elev= 30
  4420.2  377.32  4454.3  374.37  4461.5  374.96  4468.5  373.75  4489.8  374.25
  4517.8   372.8  4574.7  370.16  4609.9  367.32  4638.2   367.3  4647.7  366.38
  4730.1   364.3  4799.3   361.2  4857.7  360.11  4912.5  359.85  4917.9   358.9
  4978.1  359.02  4988.1  358.19  4997.5  359.07  5127.4  360.21  5222.1  361.74
  5227.4  361.12    5307  362.53  5312.3  361.94    5472     365  5734.1  376.07
  5741.5  377.09  5869.1  383.08    5912  386.31  5932.9  386.64  6008.4  390.89
#Mann= 6 ,-1 , 0
  4420.2     .08       0  4517.8      .1       0  4647.7     .08       0
  4799.3      .1       0  4857.7     .07       0  5127.4      .1       0
Bank Sta=4857.7,5127.4
XS Rating Curve= 0 ,0
Exp/Cntr=0.3,0.1

Type RM Length L Ch R = 1 ,12570   ,71,71,71
BEGIN DESCRIPTION:
UNT 005 IN RACR 26.0
END DESCRIPTION:
XS GIS Cut Line= 3
      2205137.75     13237896.83      2205537.72     13237546.85
      2206337.69     13236746.88
#Sta/Elev= 30
  4445.1  374.23  4501.5   372.6  4622.1  366.31    4736  363.05  4771.1  363.04
  4779.7  362.26    4941  357.16  4948.6   357.8  4962.8   356.5  4980.1  356.74
  4990.5  355.61  5033.1  357.86  5103.8  358.07  5132.1  359.32  5146.3  358.67
  5245.3  359.91  5273.6   361.3    5316  361.66  5372.5  363.54  5400.8   365.2
  5429.1  365.51  5471.5  367.66  5528.1  369.15  5683.7  376.23  5881.7  386.02
  5909.9  388.19  5938.2   388.8  6051.4  393.85  6065.5  395.29  6107.9  396.45
#Mann= 4 ,-1 , 0
  4445.1     .08       0  4779.7      .1       0  4948.6     .07       0
  5033.1      .1       0
Bank Sta=4948.6,5033.1
XS Rating Curve= 0 ,0
Exp/Cntr=0.3,0.1

Type RM Length L Ch R = 1 ,12499   ,82,82,82
BEGIN DESCRIPTION:
Mapping XS 2cffae9f
END DESCRIPTION:
XS GIS Cut Line= 4
       2204815.5     13238152.21      2205367.59     13237766.78
      2205645.37     13237537.62      2206252.82     13236891.98
#Sta/Elev= 30
  4009.6  383.11    4023   381.5  4073.3   382.3  4151.3  381.29  4166.1  379.89
    4187   380.7  4201.9  379.04    4208  380.17  4275.2  378.95  4352.4  376.16
  4597.7  365.18  4610.1  366.01  4756.7  361.64  4838.7  359.49  4860.8  362.32
  4881.6   362.4  4889.5  358.94    4896  357.91  4916.8  353.61    4939  352.04
    4995  351.36    5038  353.63  5059.2   357.2  5066.5  357.77  5073.4  361.11
  5087.5  361.69  5123.2   357.5  5335.2  362.11  5660.9   375.8  5929.5  389.28
#Mann= 6 ,-1 , 0
  4009.6      .1       0  4275.2     .05       0  4352.4     .08       0
  4756.7      .1       0    4896     .07       0  5059.2      .1       0
#XS Ineff= 2 , 0
         4878.57  362.46 5089.29           361.8
Permanent Ineff=
       F       F
Bank Sta=4896,5066.5
XS Rating Curve= 0 ,0
Exp/Cntr=0.3,0.1

Type RM Length L Ch R = 1 ,12417   ,70,70,70
BEGIN DESCRIPTION:
Mapping XS 36fc727f
END DESCRIPTION:
XS GIS Cut Line= 5
      2204763.43     13238259.84       2205579.4     13237673.03
      2205645.37     13237648.73      2205687.04     13237603.59
      2206293.23     13236952.36
#Sta/Elev= 30
  3880.6  382.58  3987.5  380.45  4035.6  379.91    4065  378.12  4088.4  378.68
  4115.3  376.87  4136.2   377.8  4144.6  376.74  4266.3  375.51  4396.6  371.54
  4560.7  365.73  4675.1   362.6  4735.4  361.88  4788.1  359.45  4832.2  359.06
  4838.4  360.41  4867.8  360.71    4874  362.45  4914.3  362.43  4972.9  359.84
    4987  357.03    5001  354.53  5008.6  356.66  5022.8  357.18  5036.9  359.71
  5043.8  357.14  5051.1  358.03  5107.8  357.15  5340.8  362.39  5907.1  388.18
#Mann= 9 ,-1 , 0
  3880.6     .05       0  3987.5      .1       0  4088.4     .05       0
  4396.6     .08       0  4560.7      .1       0  4675.1     .08       0
  4735.4      .1       0    4987     .07       0  5022.8      .1       0
Bank Sta=4987,5022.8
XS Rating Curve= 0 ,0
Exp/Cntr=0.3,0.1

Type RM Length L Ch R = 1 ,12347   ,378,378,378
BEGIN DESCRIPTION:
Mapping XS 87302696
END DESCRIPTION:
XS GIS Cut Line= 3
      2204909.27     13238322.33      2205773.84     13237620.95
      2206303.89     13237025.08
#Sta/Elev= 30
  3938.1  375.25  4210.8  371.65  4396.2  367.72  4402.6  368.46  4411.1  367.29
  4502.7  365.71  4538.5     364  4658.5   362.6  4722.3  362.18  4778.6  359.58
  4886.9  357.96  4907.7  358.67  4922.1  357.27  4957.3  356.63    4986  357.16
  5000.1     354  5014.8   355.5  5050.7  356.54  5191.3  358.24  5390.3  364.48
  5411.2  366.31  5425.4  365.88  5545.8  371.02  5623.6  376.12  5729.8   379.9
  5737.3  381.28  5758.2  381.16  5765.7  382.64    5836     385  5848.9  386.34
#Mann= 6 ,-1 , 0
  3938.1     .05       0  4411.1      .1       0  4658.5     .08       0
  4778.6      .1       0    4986     .07       0  5050.7      .1       0
Bank Sta=4986,5050.7
XS Rating Curve= 0 ,0
Exp/Cntr=0.3,0.1

Type RM Length L Ch R = 1 ,11969   ,288,288,288
BEGIN DESCRIPTION:
UNT 005 IN RACR 25.0
END DESCRIPTION:
XS GIS Cut Line= 4
       2205890.6     13238392.46      2205964.72      13238048.8
       2206207.3     13237368.26      2206281.42     13237253.69
#Sta/Elev= 30
  4374.1  373.06  4492.1  367.86  4592.5  363.72  4620.8  363.66  4714.2  359.31
  4808.2  356.97  4940.1  354.69    4957  355.51  4962.3  354.93  4987.8  355.19
  4993.1  352.71  5003.5  350.71  5006.8  351.21  5013.3  354.66  5049.4  354.44
  5131.1  356.21  5167.4  358.38  5247.9   360.4  5279.8  362.22  5316.2  362.74
  5341.7  364.75  5377.8  365.56  5403.3  368.19    5457  370.97  5493.2     372
  5508.4  373.91  5529.5  373.89  5544.7  375.96  5550.6  375.19  5584.6  377.08
#Mann= 5 ,-1 , 0
  4374.1     .05       0  4492.1     .08       0  4592.5      .1       0
  4987.8     .07       0  5013.3      .1       0
Bank Sta=4987.8,5013.3
XS Rating Curve= 0 ,0
Exp/Cntr=0.3,0.1

Type RM Length L Ch R = 1 ,11681   ,354,354,354
BEGIN DESCRIPTION:
UNT 005 IN RACR 24.0
END DESCRIPTION:
XS GIS Cut Line= 4
      2206079.25     13238459.86      2206267.94     13238143.14
      2206382.49     13237590.61      2206416.17     13237307.65
#Sta/Elev= 30
    4302  372.89  4317.1  373.15  4392.3   368.6  4456.8  366.35  4479.4  366.48
  4506.7  363.95    4515  364.26  4559.3  361.72  4693.3  356.84  4809.8  354.53
    4912  354.42    4939  353.44  4983.5  353.39  4989.2  349.88  4994.3  352.12
  5003.6  348.88  5006.9  349.38  5014.1  352.95  5039.3  353.04  5184.7  360.69
  5218.3  361.07  5240.3  362.99  5322.9  365.98  5359.6  368.51  5389.8  368.85
  5399.9  370.35  5410.5  370.25  5460.3  372.93  5488.1  375.51  5519.9  376.94
#Mann= 4 ,-1 , 0
    4302     .08       0  4392.3      .1       0  4983.5     .07       0
  5014.1      .1       0
Bank Sta=4983.5,5014.1
XS Rating Curve= 0 ,0
Exp/Cntr=0.3,0.1

Type RM Length L Ch R = 1 ,11327   ,470,470,470
BEGIN DESCRIPTION:
UNT 005 IN RACR 23.0
END DESCRIPTION:
XS GIS Cut Line= 4
      2206166.89     13238628.26       2206544.2     13238311.59
      2206712.65     13237691.68      2206678.96     13237374.95
#Sta/Elev= 30
  4072.2  375.11  4142.9  373.21  4148.8  373.16  4173.3  372.58  4187.7  370.59
  4216.3  369.16  4280.2  366.71  4399.7  362.79  4407.5  361.94    4414  362.44
  4436.1  360.87  4442.6  361.34  4596.4  355.93  4631.1  355.96  4642.2  354.92
  4715.8  352.78  4978.8  351.66  4984.2  351.18  4994.3  347.44  4997.6  347.94
  5004.9  351.04  5013.4  352.22  5053.2  351.65  5098.2  354.45  5160.4  356.17
  5252.3  360.24  5282.4  362.77    5383  366.74  5513.7  374.58  5525.7   374.6
#Mann= 6 ,-1 , 0
  4072.2     .05       0  4142.9     .08       0  4148.8     .05       0
  4280.2      .1       0  4978.8     .07       0  5013.4      .1       0
Bank Sta=4978.8,5013.4
XS Rating Curve= 0 ,0
Exp/Cntr=0.3,0.1

Type RM Length L Ch R = 1 ,10857   ,433,433,433
BEGIN DESCRIPTION:
UNT 005 IN RACR 22.0
END DESCRIPTION:
XS GIS Cut Line= 4
      2206773.28     13238938.27      2206988.91     13238426.14
      2207116.94     13237826.45      2206887.86     13237354.82
#Sta/Elev= 30
  4149.7  370.45  4199.9  369.21    4282  365.96  4292.3  366.33  4300.3  365.18
  4606.8  355.41  4628.6   355.6  4650.3  354.37  4827.3  351.17    4858  350.06
  4898.9  349.77  4909.2   349.1  4964.2  349.09    4991  348.13  5000.9  345.75
  5013.8  349.34  5031.9  349.64  5052.3  348.74  5058.2   349.8  5072.8  349.43
  5164.8   350.2  5321.1  352.97  5534.6  359.99  5579.7   362.1  5596.1  362.26
  5602.3   363.2  5751.7   368.8  5760.2  368.44  5773.9  369.78  5842.9  371.85
#Mann= 3 , 0 , 0
  4149.7      .1       0  4964.2     .07       0  5013.8      .1       0
Bank Sta=4964.2,5013.8
XS Rating Curve= 0 ,0
Exp/Cntr=0.3,0.1

Type RM Length L Ch R = 1 ,10424   ,500,500,500
BEGIN DESCRIPTION:
UNT 005 IN RACR 21.0
END DESCRIPTION:
XS GIS Cut Line= 3
       2207480.8     13238938.25      2207460.58     13237934.26
      2207393.27     13237261.11
#Sta/Elev= 30
    4270  370.72  4311.4  369.69  4371.4  366.93  4401.4  366.48  4471.4  363.38
  4511.4   362.6  4531.4  360.94  4561.5  360.33  4591.5  358.55  4681.5  356.19
  4701.5  354.56  4721.5  354.36  4741.5  352.95  4951.5  346.49  4981.5  346.66
  4991.5  345.72  5001.3  343.47  5011.5  345.34  5021.5  345.18  5031.5  346.32
  5111.6  347.89  5402.2  350.74  5412.3  351.69  5502.7  353.05  5643.4  357.17
  5656.6  357.01  5663.5  357.83  5733.9   359.4  5804.2  362.35  5950.7  366.97
#Mann= 3 , 0 , 0
    4270      .1       0  4981.5     .07       0  5031.5      .1       0
Bank Sta=4981.5,5031.5
XS Rating Curve= 0 ,0
Exp/Cntr=0.3,0.1

Type RM Length L Ch R = 1 ,9924    ,398,398,398
BEGIN DESCRIPTION:
UNT 005 IN RACR 20.0
END DESCRIPTION:
XS GIS Cut Line= 4
      2208067.01     13238918.04      2208019.84     13238500.26
      2207844.65      13237765.8      2207521.98     13237234.74
#Sta/Elev= 30
  4318.3   368.7  4353.8  366.85  4360.7  367.31  4430.2  364.14  4450.5  361.58
  4530.3  360.42  4591.2  356.68  4768.7  349.75  4978.7  344.03  4984.4  341.83
  4989.5  342.64    4999  340.35  5002.3  340.85  5009.5  344.34  5242.2  344.83
  5389.9  345.99    5431  347.48  5451.6  346.82  5724.7  354.64  5730.5  354.15
    5746  355.38  5761.5   354.8  5773.4  356.38  5796.8  356.12  5935.9   361.1
  5941.8  362.06  5978.6  362.91  5984.4  362.01  6015.4  364.09  6115.2  367.11
#Mann= 4 ,-1 , 0
  4318.3     .05       0  4353.8      .1       0  4978.7     .07       0
  5009.5      .1       0
Bank Sta=4978.7,5009.5
XS Rating Curve= 0 ,0
Exp/Cntr=0.3,0.1

Type RM Length L Ch R = 1 ,9526    ,475,475,475
BEGIN DESCRIPTION:
UNT 005 IN RACR 19.0
END DESCRIPTION:
XS GIS Cut Line= 4
      2208309.58     13238904.52      2208343.27     13238439.61
      2208269.15     13237631.04      2208342.85     13237262.53
#Sta/Elev= 30
    4179  365.76  4222.1  364.79  4236.8  363.49  4246.8  363.85  4276.9  363.21
  4286.9  362.07  4307.8  361.23  4347.1  359.93  4356.4  358.95  4361.5   359.2
  4427.3  355.96  4547.6  352.45  4597.8  349.62    4652  349.16  4698.1  347.22
  4818.6  344.67  4858.8   344.7  4969.2  342.38  4982.1  342.59  4989.3  339.95
  4999.1  337.98  5002.4  338.48  5009.4   341.4  5029.5  342.44  5059.6  342.05
  5180.1  343.34  5280.5  345.68  5370.9  345.93    5476  347.77  5832.9  359.53
#Mann= 4 ,-1 , 0
    4179     .05       0  4307.8      .1       0  4982.1     .07       0
  5029.5      .1       0
Bank Sta=4982.1,5029.5
XS Rating Curve= 0 ,0
Exp/Cntr=0.3,0.1

Type RM Length L Ch R = 1 ,9051    ,338,338,338
BEGIN DESCRIPTION:
UNT 005 IN RACR 18.0
END DESCRIPTION:
XS GIS Cut Line= 3
      2209077.74     13238810.24      2208828.41     13238325.06
      2208599.31     13237253.67
#Sta/Elev= 30
  4011.2  357.86  4112.5   355.2  4171.1  353.81  4176.7  352.99  4215.4  352.32
  4319.7  348.48  4481.6  345.39  4556.7  345.35    4698  342.91  4738.9  343.26
  4749.2  342.54  4769.6  342.09  4780.1  342.62    4839  340.85  4873.9  341.34
  4918.3  340.45  4953.7  340.69  4974.1   339.4  4984.4  339.74  5004.6  335.49
  5007.8  335.99  5012.1  338.81  5017.2  338.75  5025.3  340.66  5061.6  340.01
    5106  340.42  5260.5  343.63  5372.9  348.45  5535.9  353.52  5652.3  358.47
#Mann= 6 ,-1 , 0
  4011.2     .05       0  4112.5      .1       0  4319.7     .05       0
    4839      .1       0  4984.4     .07       0  5025.3      .1       0
Bank Sta=4984.4,5025.3
XS Rating Curve= 0 ,0
Exp/Cntr=0.3,0.1

Type RM Length L Ch R = 1 ,8713    ,428,428,428
BEGIN DESCRIPTION:
UNT 005 IN RACR 17.0
END DESCRIPTION:
XS GIS Cut Line= 3
      2209237.72     13238546.87      2209037.72     13237746.85
       2208837.7     13237346.81
#Sta/Elev= 30
  4197.6  354.63    4319  349.42  4460.7  344.18  4496.5  342.75  4601.7  340.66
  4640.9  340.43  4661.5  340.97  4692.4  339.82  4760.6  339.29  4872.3  339.22
  4921.7  339.22  4957.8  337.86    4981  337.61    4999  336.44  5001.2  334.45
  5003.9  333.95  5007.2  334.45  5011.9  337.83  5044.6  337.87  5097.7     340
  5111.7  339.81  5125.7  340.61    5134  340.49  5201.1  343.12  5237.5  343.94
  5254.2  345.39  5335.3  346.88  5371.6  348.02  5388.4   349.3  5469.5  352.03
#Mann= 8 ,-1 , 0
  4197.6     .05       0    4319      .1       0  4460.7     .05       0
  4601.7      .1       0  4760.6     .05       0  4872.3      .1       0
    4981     .07       0  5011.9      .1       0
Bank Sta=4981,5011.9
XS Rating Curve= 0 ,0
Exp/Cntr=0.3,0.1

Type RM Length L Ch R = 1 ,8285    ,470,470,470
BEGIN DESCRIPTION:
UNT 005 IN RACR 16.0
END DESCRIPTION:
XS GIS Cut Line= 3
      2209987.74     13238446.88      2209437.72     13237646.85
       2209187.7     13237296.83
#Sta/Elev= 30
  4018.8  356.47  4068.2  354.16  4104.1  353.39  4118.9  352.18  4148.7  351.59
  4184.6  349.93  4199.5  350.06  4220.4  348.78  4342.9  344.51  4384.8  344.27
  4486.3  340.32    4558  339.12  4572.9  338.26  4746.1  336.35  4838.8  337.07
  4874.6   335.3  4889.5   336.1  4925.4  335.15  4982.2  334.95  4986.4   334.2
  5026.5  335.99  5139.6  338.16  5169.1  339.18    5190  340.81  5198.6  340.29
  5269.8  343.06  5284.6  343.12  5341.1  346.17  5382.9  347.38  5419.8  349.73
#Mann= 3 , 0 , 0
  4018.8     .05       0  4889.5     .07       0  5026.5      .1       0
Bank Sta=4889.5,5026.5
XS Rating Curve= 0 ,0
Exp/Cntr=0.3,0.1

Type RM Length L Ch R = 1 ,7815    ,473,473,473
BEGIN DESCRIPTION:
UNT 005 IN RACR 15.0
END DESCRIPTION:
XS GIS Cut Line= 3
      2210487.71     13238296.84      2209837.72     13237496.85
      2209437.75     13237096.88
#Sta/Elev= 30
  3977.7  358.17  4155.8  350.56  4176.6  350.31  4183.8  350.94  4205.4  348.64
  4254.9   345.7  4454.4  338.03  4539.4  335.74  4545.8  336.27  4568.1  334.98
  4617.7  333.88  4731.2  333.44    4752  334.34  4766.4  333.47  4802.6  333.83
  4815.9  334.55    4923  333.89  4986.9  332.82    5001  331.75  5005.2  332.53
  5036.7  332.62  5079.2  334.01  5135.7  335.98  5206.4  336.43  5234.7  338.76
    5263  337.88  5291.3   339.3    5362  340.94  5432.7  344.48  5574.1  348.56
#Mann= 4 ,-1 , 0
  3977.7     .05       0  4802.6      .1       0    4923     .07       0
  5079.2      .1       0
Bank Sta=4923,5079.2
XS Rating Curve= 0 ,0
Exp/Cntr=0.3,0.1

Type RM Length L Ch R = 1 ,7342    ,439,439,439
BEGIN DESCRIPTION:
UNT 005 IN RACR 14.0
END DESCRIPTION:
XS GIS Cut Line= 3
      2210537.73     13238246.89      2210287.72     13237446.85
      2209487.71     13236846.85
#Sta/Elev= 30
  4160.4  356.81  4286.2  351.34  4328.1  348.48  4408.8  344.78  4502.9  340.78
  4607.4  336.44    4712  333.08  4797.5  332.08  4841.4  331.22  4915.7  331.29
  4917.4  331.36  4995.7     330  5005.9  330.91  5048.6  331.38    5185  331.78
  5205.9  332.68  5241.3  331.86  5255.9  332.79  5362.1  332.56  5476.7  335.09
    5594  339.22  5719.8  343.93  5762.1  346.51  5798.6  347.39  5891.3  351.47
  5905.9  352.84  5941.3  353.77  5955.9  355.09  5970.5  354.81  5998.6  356.49
#Mann= 9 ,-1 , 0
  4160.4     .05       0  4408.8      .1       0  4502.9     .05       0
  4607.4      .1       0  4797.5     .05       0  4915.7     .07       0
  5048.6      .1       0    5594     .05       0  5719.8      .1       0
Bank Sta=4917.4,5048.6
XS Rating Curve= 0 ,0
Exp/Cntr=0.3,0.1

Type RM Length L Ch R = 1 ,6903    ,425,425,425
BEGIN DESCRIPTION:
UNT 005 IN RACR 13.0
END DESCRIPTION:
XS GIS Cut Line= 3
      2211037.72     13237646.85      2210637.72     13237246.85
      2209837.71     13236546.85
#Sta/Elev= 30
  4410.4  343.65  4551.8  339.75    4665  337.98  4801.4  333.99  4914.2  331.23
  4961.9  329.45  4983.2  328.18  5011.7  327.87  5018.1  327.21  5054.4   329.1
  5082.4  328.61  5146.4  329.32  5273.6  328.57  5316.3  329.22  5351.5  328.74
  5457.8  328.85  5585.9   329.8  5663.7  331.46  5670.4  331.02  5698.8  331.51
  5727.3  332.83  5748.2  332.88  5784.3  334.36  5805.1  334.39  5833.6  335.91
  5862.1  336.32  5939.9  338.95  5968.4  340.68  5982.6  340.64  6039.1   343.3
#Mann= 5 ,-1 , 0
  4410.4      .1       0  4801.4     .05       0  4914.2      .1       0
  4961.9     .07       0  5054.4      .1       0
Bank Sta=4961.9,5054.4
XS Rating Curve= 0 ,0
Exp/Cntr=0.3,0.1

Type RM Length L Ch R = 1 ,6478    ,499,499,499
BEGIN DESCRIPTION:
UNT 005 IN RACR 12.0
END DESCRIPTION:
XS GIS Cut Line= 3
      2211587.75     13237296.87      2210787.72     13236846.85
      2209987.75     13236296.88
#Sta/Elev= 30
  4085.4  355.35  4140.4  353.23  4263.7  348.11  4438.9  340.56  4498.2  338.78
  4649.9  332.54    4806  329.84  4833.4  328.53  4908.7  327.49  4914.4  327.31
  4995.3  325.72  5000.2   325.1  5039.7  327.04  5148.1  326.34  5233.9  327.57
  5246.8  327.06  5282.7   327.5  5355.2  326.91  5485.7  327.43  5506.7  328.07
  5549.4  327.73  5599.3  329.21  5614.2  328.62    5644  329.79  5679.9   330.1
  5802.3  335.27  5816.4  335.11  5945.7  339.67  5960.6  340.91  5974.1  340.75
#Mann= 5 ,-1 , 0
  4085.4     .05       0  4140.4      .1       0  4263.7     .05       0
  4908.7     .07       0  5039.7      .1       0
Bank Sta=4914.4,5039.7
XS Rating Curve= 0 ,0
Exp/Cntr=0.3,0.1

Type RM Length L Ch R = 1 ,5979    ,478,478,478
BEGIN DESCRIPTION:
UNT 005 IN RACR 11.0
END DESCRIPTION:
XS GIS Cut Line= 3
       2211437.7     13236946.84      2211037.72     13236546.85
       2210237.7     13235846.84
#Sta/Elev= 30
  4436.4  340.09  4719.2  329.04  4916.6  324.88  4973.8  324.58  4998.3  323.36
  5015.8  324.43  5193.3  324.92  5200.9   325.4  5256.9   324.5  5264.5  324.69
  5271.1  326.02    5293  324.22    5385  325.72  5505.6  326.52  5547.3  327.84
  5583.4  327.72  5626.1  328.74  5767.5  329.86  5916.5  332.78  5930.8  332.15
  5980.1   333.8    6001  333.96  6008.6  332.54  6022.8  334.22  6029.5   334.1
  6037.1  335.64  6043.7  335.81    6058   338.6  6061.8  340.95  6065.1  340.95
#Mann= 4 ,-1 , 0
  4436.4     .05       0  4916.6      .1       0  4973.8     .07       0
  5015.8      .1       0
Bank Sta=4973.8,5015.8
XS Rating Curve= 0 ,0
Exp/Cntr=0.3,0.1

Type RM Length L Ch R = 1 ,5501    ,416,416,416
BEGIN DESCRIPTION:
UNT 005 IN RACR 10.0
END DESCRIPTION:
XS GIS Cut Line= 4
      2211584.87      13236906.3        2211461.     13236571.38
      2210924.17      13235699.6      2210488.27     13235098.52
#Sta/Elev= 30
    4155  340.75  4251.7   337.1  4441.4  328.56    4599  324.27  4656.9  323.66
  4693.6  324.05  4720.8  323.15  4794.1  323.65  4940.2  322.69  4989.3   322.1
  5004.5  321.03  5010.6  321.76  5047.3  322.58  5362.1  325.63  5374.7  325.91
  5383.3  326.93    5586  329.66  5713.6  332.61  5742.9  332.48  5757.6  333.65
  5763.8  333.09  5793.2  334.19  5835.8  334.43  5971.6  337.16  6121.8  340.83
  6151.2  342.19  6222.3  342.89  6251.7  344.35  6272.5  344.19  6278.4  344.88
#Mann= 4 ,-1 , 0
    4155     .05       0  4441.4      .1       0  4940.2     .07       0
  5047.3      .1       0
Bank Sta=4940.2,5047.3
XS Rating Curve= 0 ,0
Exp/Cntr=0.3,0.1

Type RM Length L Ch R = 1 ,5085    ,376,376,376
BEGIN DESCRIPTION:
UNT 005 IN RACR 9.0
END DESCRIPTION:
XS GIS Cut Line= 4
      2211782.18     13236860.39      2211786.77     13236594.32
      2211447.23     13235607.84      2211153.56     13235093.91
#Sta/Elev= 30
  4089.4  338.67  4152.9  336.46  4242.5  331.47    4303  330.05  4394.3  325.58
  4456.7  323.96  4644.1  321.66  4831.4  322.24  4945.1  321.44  4951.1  320.94
  4982.3  320.66  4997.7  319.01  5008.2   320.5  5039.4  320.88  5044.7  320.84
  5114.3  321.94  5241.2  321.92  5346.4  323.81  5368.1  325.18  5471.6  327.42
    5568  331.92  5618.8  333.14  5627.1  334.28    5780   338.8  5825.7   341.6
  5860.6  342.08  5890.5  343.92  5912.1  343.32  5949.5  345.65  5990.7  345.73
#Mann= 4 ,-1 , 0
  4089.4     .05       0  4242.5      .1       0  4951.1     .07       0
  5044.7      .1       0
Bank Sta=4945.1,5039.4
XS Rating Curve= 0 ,0
Exp/Cntr=0.3,0.1

Type RM Length L Ch R = 1 ,4709    ,531,531,531
BEGIN DESCRIPTION:
UNT 005 IN RACR 8.0
END DESCRIPTION:
XS GIS Cut Line= 4
      2212199.71     13236910.89      2212236.42     13236456.67
      2211717.94     13235456.42      2211392.47     13234952.17
#Sta/Elev= 30
  3832.4  336.19  3997.9  329.63  4120.2  326.24  4127.4  324.84  4157.5  325.57
  4366.8  321.62  4637.1  318.39  4886.7  320.97  4963.7  319.74  4997.2  317.46
  5013.8  319.23  5052.4  319.29  5058.1  319.54  5146.6  319.61  5168.7  318.77
  5190.8  319.59  5207.3  318.19  5257.2  318.81    5318  321.03  5334.5  322.08
  5340.1  323.43  5369.2  323.28  5567.4  331.23    5770  337.39  5791.2  339.16
  5878.4  342.07  5936.3  343.13  5942.3   344.2  5949.8  343.46  6014.9  346.44
#Mann= 3 ,-1 , 0
  3832.4      .1       0  4963.7     .07       0  5052.4      .1       0
Bank Sta=4963.7,5058.1
XS Rating Curve= 0 ,0
Exp/Cntr=0.3,0.1

Type RM Length L Ch R = 1 ,4178    ,353,353,353
BEGIN DESCRIPTION:
UNT 005 IN RACR 7.0
END DESCRIPTION:
XS GIS Cut Line= 4
      2212718.17     13236686.05      2212475.01     13236300.67
      2211942.77     13235194.89      2211543.57     13234827.81
#Sta/Elev= 30
  3524.4  334.06  3726.2  327.62  3771.8  327.64  3793.2  326.18  3966.2   322.7
  4017.6  320.69  4106.4  318.94  4264.7  317.19  4317.3   317.4  4354.9  316.39
    4406  317.46  4513.6  317.24    4587  318.46  4649.3  318.03  4716.8  318.96
    4850  319.35  4983.1  318.38  4999.8  317.44  5016.4  318.45  5022.5  318.46
  5141.1  323.15  5158.2  322.83  5393.3  331.58    5450  332.85  5492.6  335.21
  5527.7  335.48  5535.1  336.67  5690.5  343.05  5704.7  344.33  5749.6   345.3
#Mann= 3 ,-1 , 0
  3524.4      .1       0  4983.1     .07       0  5022.5      .1       0
Bank Sta=4983.1,5016.4
XS Rating Curve= 0 ,0
Exp/Cntr=0.3,0.1

Type RM Length L Ch R = 1 ,3825    ,596,596,596
BEGIN DESCRIPTION:
UNT 005 IN RACR 6.0
END DESCRIPTION:
XS GIS Cut Line= 3
      2212787.71     13236496.83      2212387.72     13235296.85
      2211587.69     13234496.83
#Sta/Elev= 30
  3659.5  331.99  3838.7  324.84  4186.5  315.51  4270.9   314.7  4418.4  315.43
  4460.3   314.2  4471.1  315.14  4629.2  315.99  4650.3  316.94  4892.8  316.67
  4921.8  315.19  4995.1  315.26  5023.4  316.47  5037.5  317.95    5080  317.74
  5108.2  319.06  5207.2  319.71  5334.5  323.83  5405.2  324.94  5433.5  327.06
  5518.4  328.31  5625.1  332.52  5679.5  334.73  5767.3     338  5837.4  341.23
  5857.8   342.2  5871.9  344.22  5900.2  344.09  5967.3  347.04  6055.8  351.57
#Mann= 8 ,-1 , 0
  3659.5     .16       0  4892.8     .07       0  5023.4      .1       0
  5625.1     .05       0  5679.5      .1       0  5767.3     .05       0
  5837.4      .1       0  5967.3     .05       0
Bank Sta=4892.8,5023.4
XS Rating Curve= 0 ,0
Exp/Cntr=0.3,0.1

Type RM Length L Ch R = 1 ,3229    ,429,429,429
BEGIN DESCRIPTION:
UNT 005 IN RACR 5.0
END DESCRIPTION:
XS GIS Cut Line= 3
      2213080.65     13236429.09      2212805.37     13235282.07
      2212516.79      13234801.1
#Sta/Elev= 30
  3881.1   333.3  4222.8  318.61  4325.6  315.22    4377  315.13  4418.2   313.3
  4473.4  313.51  4487.1  312.31  4510.3  311.12  4531.3  311.61  4551.6  309.85
  4572.4  310.91  4646.6   311.1  4706.1  313.53  4963.2  315.12  4987.6  313.66
  5004.4     313  5024.5  314.71  5029.6  314.93  5035.2  315.81  5063.4  314.18
    5257  315.92  5498.5   318.1  5521.6  319.57  5529.9   321.9  5544.3  318.92
  5572.6  319.79  5588.2   322.7  5603.2  328.38  5609.6   328.5  5621.6  323.31
#Mann= 7 ,-1 , 0
  3881.1     .16       0  4487.1     .16       0  4987.6     .07       0
  5024.5     .16       0    5257     .05       0  5498.5      .1       0
  5544.3     .05       0
Bank Sta=4963.2,5029.6
XS Rating Curve= 0 ,0
Exp/Cntr=0.3,0.1

Type RM Length L Ch R = 1 ,2800    ,384,384,384
BEGIN DESCRIPTION:
UNT 005 IN RACR 4.0
END DESCRIPTION:
XS GIS Cut Line= 4
      2213305.49     13236452.05      2213287.14     13235984.08
      2213199.96     13234983.83      2212792.15     13234337.74
#Sta/Elev= 30
  3885.1  332.38  3955.6  328.76  4000.4  328.21  4070.4  323.15  4142.5  321.25
  4200.5  318.25  4349.5  313.34  4501.2  311.52  4561.2     309  4571.5  309.88
  4681.9  311.01  4942.9  312.43    4963  311.09  5023.2  312.17  5043.3  313.99
  5135.3  313.15  5203.9  312.38  5486.7  313.97  5621.2  317.48  5684.3  319.29
  5711.4  322.69  5720.5  322.38  5726.7  320.57  5747.9  320.78  5778.4  322.73
  5850.6  325.25  5863.2  324.76  5893.8  326.84  5988.8  330.03  6121.5  334.73
#Mann= 7 ,-1 , 0
  3885.1      .1       0  4142.5     .05       0  4942.9     .07       0
  5023.2      .1       0  5135.3     .05       0  5621.2      .1       0
  5988.8     .05       0
Bank Sta=4942.9,5023.2
XS Rating Curve= 0 ,0
Exp/Cntr=0.3,0.1

Type RM Length L Ch R = 1 ,2416    ,616,616,616
BEGIN DESCRIPTION:
UNT 005 IN RACR 3.0
END DESCRIPTION:
XS GIS Cut Line= 5
      2213580.78     13236520.92      2213750.56     13235993.25
      2213484.43     13234859.94      2213016.43     13234346.05
      2212878.75     13234212.96
#Sta/Elev= 30
  3792.5  329.47  3811.8  328.28  3960.8  321.99  4080.4  318.77  4121.2  318.81
    4238  314.24  4445.8   310.4  4671.6  308.32  4805.3  310.33  4959.4  310.27
  4969.7  309.82  5000.5  309.06 5014.03  310.34  5031.3  313.31    5042  313.56
  5062.1  311.94  5090.5  311.73  5349.8  310.69  5386.5  311.33  5401.1  312.94
    5434  311.69  5567.7  315.02  5730.5  316.15  5907.4  320.06  5949.4  323.67
  5971.1  321.34    5992  321.93  6077.1  326.76  6148.1  328.15  6397.5   337.6
#Mann= 5 ,-1 , 0
  3792.5      .1       0  3811.8     .05       0  4969.7     .07       0
 5014.03      .1       0  5090.5     .05       0
Bank Sta=4959.4,5014.03
XS Rating Curve= 0 ,0
Exp/Cntr=0.3,0.1

Type RM Length L Ch R = 1 ,1800    ,547,547,547
BEGIN DESCRIPTION:
UNT 005 IN RACR 2.0
END DESCRIPTION:
XS GIS Cut Line= 4
      2213970.78     13236598.94      2214145.15     13236007.02
      2214039.62     13234905.83      2213787.85      13234260.4
#Sta/Elev= 30
  4061.5  329.82  4230.5  322.43  4261.7  322.62  4324.3  319.77  4571.1  312.97
  4703.9   309.4  4796.9  308.68  4839.5  307.51  4980.1  308.21  5021.9  307.24
  5030.3     309  5040.4  310.95  5050.4  310.87  5070.5  308.59  5090.6  307.97
    5232  306.56  5412.1  308.24  5848.1     308    5934  309.53  5976.9  312.52
  6009.1  311.89  6202.3  317.89  6239.8  321.05  6266.5  320.48  6277.5  321.79
  6309.7  322.42  6356.1  326.62  6374.1  324.33  6435.8   326.9  6477.6  329.19
#Mann= 6 ,-1 , 0
  4061.5      .1       0  4571.1     .05       0  4796.9     .07       0
  5030.3     .05       0  6239.8      .1       0  6435.8     .05       0
#XS Ineff= 2 , 0
                         5047.72          311.01
Permanent Ineff=
       F       F
Bank Sta=4796.9,5030.3
XS Rating Curve= 0 ,0
Exp/Cntr=0.3,0.1

Type RM Length L Ch R = 1 ,1253    ,919,919,919
BEGIN DESCRIPTION:
Mapping XS 6e6f3506
END DESCRIPTION:
XS GIS Cut Line= 5
      2214429.61       13236732.      2214585.62      13236250.2
      2214613.15     13235658.31      2214278.21     13234937.94
      2213865.42     13234231.61
#Sta/Elev= 30
  4128.9  334.55  4176.5  332.29  4186.9  332.83    4292  327.24  4323.5  326.53
    4355   324.2  4386.6  324.08  4418.1  321.69  4463.5  320.14    4700  310.81
  4878.9  305.92    4959  306.24    4979  307.19 4984.07  306.44  4998.4  304.16
  5009.1  306.46  5300.6  307.46  5333.6  305.72  6197.4  307.05  6330.5  309.78
  6359.4  312.42  6382.6   312.2  6447.8  314.89  6490.8  315.47    6528   317.5
  6638.4  320.97  6688.4  322.82  6704.1  325.24  6741.3  325.11  6840.4  329.23
#Mann= 7 ,-1 , 0
  4128.9      .1       0  4463.5     .05       0    4700      .1       0
 4984.07     .07       0  5009.1      .1       0  5333.6     .05       0
  6638.4      .1       0
Bank Sta=4984.07,5009.1
XS Rating Curve= 0 ,0
Exp/Cntr=0.3,0.1
