HEC-RAS study SALT BRANCH.prj: SALT BRANCH Base Level Engineering

--- SALT BRANCH.g01 (geometry) --- (continued)

Type RM Length L Ch R = 1 ,65107   ,475,475,475
BEGIN DESCRIPTION:
SALT BRANCH 95.0
END DESCRIPTION:
XS GIS Cut Line= 2
      2219828.77     13309280.51      2221010.46      13308311.8
#Sta/Elev= 30
  3999.7  264.15  4101.7  260.34  4186.3  258.43  4278.9  257.94    4378  259.54
    4477  257.95  4690.9  250.39  4733.9  250.54  4761.2  248.96  4868.1   247.5
  4925.5  248.53  4960.7  247.63  4968.1  244.85  4981.5  245.31    4997  238.18
  4999.8  237.68    5003  238.18  5010.2  238.69  5018.1  242.56  5038.9  246.38
  5045.7  250.54  5131.5  258.61  5166.7  261.08  5174.6   260.8    5188  262.59
  5195.4  262.21  5230.6  265.84  5273.6  268.23  5294.4  270.38  5527.7  283.52
#Mann= 3 ,-1 , 0
  3999.7      .1       0    4997     .07       0    5003      .1       0
Bank Sta=4981.5,5038.9
XS Rating Curve= 0 ,0
Exp/Cntr=0.3,0.1

Type RM Length L Ch R = 1 ,64632   ,462,462,462
BEGIN DESCRIPTION:
SALT BRANCH 94.0
END DESCRIPTION:
XS GIS Cut Line= 3
      2220137.69     13309646.88      2220737.72     13309096.85
      2221087.73     13308696.85
#Sta/Elev= 30
  4187.3  266.79  4505.8  253.84  4647.6  250.37  4654.4  250.99  4689.6  250.59
    4697  249.83  4732.1  249.54  4796.3  247.34  4866.5  247.82  4916.5  246.26
  4965.8  247.71  4973.2  246.57    4980  242.46  4994.2  240.95    4997  236.43
  4999.8  235.93    5003  236.43  5004.6  238.29  5008.4  236.43    5015  242.45
  5022.6  246.36  5043.5  247.56  5065.3  247.36  5185.9  250.78  5468.7  265.38
  5497.2   267.6    5519  272.27  5525.7  272.44  5529.5  275.39  5532.8  275.39
#Mann= 3 ,-1 , 0
  4187.3      .1       0    4997     .07       0    5003      .1       0
Bank Sta=4973.2,5022.6
XS Rating Curve= 0 ,0
Exp/Cntr=0.3,0.1

Type RM Length L Ch R = 1 ,64170   ,429,429,429
BEGIN DESCRIPTION:
SALT BRANCH 93.0
END DESCRIPTION:
XS GIS Cut Line= 3
      2220387.73     13309896.84      2220887.72     13309496.85
      2221487.69     13308946.88
#Sta/Elev= 30
  4364.4  267.42    4450  263.57  4470.8  263.94  4478.8  262.69  4520.5  261.85
  4578.1  258.78  4598.9  259.27  4606.9   257.6  4620.5  257.86  4627.7  256.46
  4648.5  256.75  4684.5  254.45  4706.2  254.48  4712.6  253.25  4848.6  246.41
  4898.2  245.96  4940.7  246.96  4976.7  244.81  4983.1  239.83  4991.1  238.72
    4997  234.03  4999.8  233.53    5003  234.03  5008.1  234.03  5018.6  241.69
    5026  242.37  5032.8  244.51  5506.9  254.44  5683.9  261.68  5818.6  269.77
#Mann= 3 ,-1 , 0
  4364.4      .1       0    4997     .07       0    5003      .1       0
Bank Sta=4976.7,5032.8
XS Rating Curve= 0 ,0
Exp/Cntr=0.3,0.1

Type RM Length L Ch R = 1 ,63741   ,355,355,355
BEGIN DESCRIPTION:
SALT BRANCH 92.0
END DESCRIPTION:
XS GIS Cut Line= 3
      2220537.69     13310146.87      2221137.72     13309846.85
      2221637.73     13309246.84
#Sta/Elev= 30
  4357.1   267.4  4482.9  262.49    4550  258.27  4714.9  250.62  4728.9  249.09
  4849.1  244.13  4924.5  245.73  4960.9  243.77  4969.3  244.01  4983.2  241.46
    4997  235.24  4999.8  234.74    5003  235.24  5005.6  235.24  5019.6  241.52
  5025.2  242.96  5041.6  243.37  5049.4  242.54  5070.3  244.01    5177  246.97
  5240.8  246.64  5298.1  248.08  5376.2  247.67  5454.3  248.67  5482.9  249.79
  5489.4  250.92  5645.6  253.84  5674.3  255.81  5709.4  256.63    5809   262.5
#Mann= 3 ,-1 , 0
  4357.1      .1       0    4997     .07       0    5003      .1       0
Bank Sta=4969.3,5025.2
XS Rating Curve= 0 ,0
Exp/Cntr=0.3,0.1

Type RM Length L Ch R = 1 ,63386   ,323,323,323
BEGIN DESCRIPTION:
SALT BRANCH 91.0
END DESCRIPTION:
XS GIS Cut Line= 3
      2220749.33     13310317.81      2221254.52     13310187.61
      2222046.22      13309635.5
#Sta/Elev= 30
  4423.5  261.08  4442.3  259.79  4488.2  258.36  4528.9  255.68  4545.8  255.64
    4618  252.03  4638.7   252.2  4691.6  250.41  4793.6  245.72  4896.9  243.39
  4930.6  243.57  4938.2  242.82  4970.1   242.3    4991  239.26    4997   234.2
  4999.8   233.7    5003   234.2  5005.8  237.78  5011.9  238.58  5020.7  243.42
  5256.2  245.71  5422.9  249.51    5644  257.96  5702.9  261.33  5744.8   262.6
  5753.5  263.54  5831.2  266.66  5881.8  269.96  5902.7   270.1  5910.4  270.86
#Mann= 3 ,-1 , 0
  4423.5      .1       0    4997     .07       0    5003      .1       0
Bank Sta=4970.1,5020.7
XS Rating Curve= 0 ,0
Exp/Cntr=0.3,0.1

Type RM Length L Ch R = 1 ,63063   ,292,292,292
BEGIN DESCRIPTION:
SALT BRANCH 90.0
END DESCRIPTION:
XS GIS Cut Line= 3
      2220947.22     13310510.52      2221613.89     13310375.11
      2222300.59      13309891.3
#Sta/Elev= 30
  4438.8  260.65  4579.9  254.91  4602.6  253.05    4674  250.85  4838.2  242.66
  4878.1  241.68  4939.4   243.5  4969.9  242.74  4979.9  239.91    4985  235.27
  4990.3  233.52    4997  233.52  4999.8  233.02    5003  233.52  5010.7  236.47
  5035.6  236.55  5051.6  240.46  5081.1  242.77  5234.4  245.95  5356.4  246.51
  5644.6  251.35  5766.6  254.67  5796.2  255.91  5802.3  257.14  5817.1  256.86
  5858.9  259.32  5888.5  259.52  5909.4  261.54  5918.1  260.84  5959.1  263.43
#Mann= 3 ,-1 , 0
  4438.8      .1       0    4997     .07       0    5003      .1       0
Bank Sta=4969.9,5081.1
XS Rating Curve= 0 ,0
Exp/Cntr=0.3,0.1

Type RM Length L Ch R = 1 ,62771   ,499,499,499
BEGIN DESCRIPTION:
SALT BRANCH 89.0
END DESCRIPTION:
XS GIS Cut Line= 3
      2221139.98     13310682.39      2221858.68     13310599.06
      2222426.38     13310234.49
#Sta/Elev= 30
  4461.6  261.54  4539.9  257.27  4570.1  254.19  4620.4  250.73  4781.5   242.6
  4841.9  240.64  4903.9  242.75  4942.5  242.67  4987.5  240.24    4997   232.2
  4999.8   231.7    5003   232.2  5023.1   240.3  5033.1  241.72  5063.3  243.19
  5084.6  243.22  5302.8  245.61  5460.4  251.32  5475.6  252.76  5496.7   252.7
  5527.1  254.89  5533.1  254.37  5589.2  256.42  5605.7   256.3  5642.1  258.24
  5742.5   259.1  5751.1  259.89    5757  259.24  5825.5  259.45  5859.8  259.66
#Mann= 6 ,-1 , 0
  4461.6      .1       0    4997     .07       0    5003      .1       0
  5084.6     .08       0  5589.2      .1       0  5825.5     .08       0
Bank Sta=4987.5,5023.1
XS Rating Curve= 0 ,0
Exp/Cntr=0.3,0.1

Type RM Length L Ch R = 1 ,62272   ,342,342,342
BEGIN DESCRIPTION:
SALT BRANCH 88.0
END DESCRIPTION:
XS GIS Cut Line= 4
      2221202.46     13311031.36      2221733.68     13311114.69
      2221884.73     13311052.19      2222534.24     13310516.99
#Sta/Elev= 30
    4390  249.22  4426.7  247.39  4557.3  243.88  4678.8  243.14  4723.5  244.41
  4840.6  243.42  4911.9  242.38  4975.4  239.73  4984.1  238.31  4989.5  237.17
    4997  230.66  4999.8  230.16    5003  230.66  5007.8  231.98  5013.4  236.24
  5029.5   238.1  5037.3  240.52  5083.6  240.96  5139.7  238.81  5189.2  240.92
  5423.7  253.22  5444.9  255.52  5637.4  266.19  5765.1  275.02  5784.1  275.34
    5829  278.01  5864.1  278.15  5892.8  280.73  5928.4  279.87  5932.8  279.81
#Mann= 9 ,-1 , 0
    4390      .1       0  4426.7     .05       0  4723.5      .1       0
  4840.6     .05       0  4911.9      .1       0    4997     .07       0
    5003      .1       0  5784.1     .08       0  5928.4      .1       0
Bank Sta=4984.1,5029.5
XS Rating Curve= 0 ,0
Exp/Cntr=0.3,0.1

Type RM Length L Ch R = 1 ,61930   ,748,748,748
BEGIN DESCRIPTION:
SALT BRANCH 87.0
END DESCRIPTION:
XS GIS Cut Line= 4
       2221332.6     13311323.01      2221858.68      13311432.4
      2222192.02     13311281.36      2222608.66     13310875.13
#Sta/Elev= 30
  4331.6  245.57  4468.9  242.51  4569.1  241.44  4684.1  241.15  4847.5  242.67
  4893.5  240.92  4941.1  238.69  4977.7  238.17  4987.3  236.22    4997  230.04
  4999.8  229.54    5003  230.04  5021.6  236.87  5032.6  239.34  5090.6  237.72
  5175.3  242.32  5211.6  242.55  5229.2  243.38  5242.2  245.14  5263.3  245.37
  5277.5  246.71  5447.2  254.79  5546.2  260.66  5588.8  264.17  5659.4   267.2
  5689.6   269.5  5701.8  271.74    5723  272.88  5730.1  274.18  5816.8   280.2
#Mann= 6 ,-1 , 0
  4331.6     .05       0  4893.5      .1       0    4997     .07       0
    5003      .1       0  5588.8     .08       0  5689.6      .1       0
Bank Sta=4977.7,5032.6
XS Rating Curve= 0 ,0
Exp/Cntr=0.3,0.1

Type RM Length L Ch R = 1 ,61182   ,652,652,652
BEGIN DESCRIPTION:
SALT BRANCH 85.0
END DESCRIPTION:
XS GIS Cut Line= 3
      2221154.81     13311644.09      2221835.04     13312118.19
      2223214.42     13312090.74
#Sta/Elev= 30
  3938.9  257.17    3979  258.05  4007.2  256.56  4022.1  257.13  4251.5  247.33
  4478.8  245.02  4611.9  245.74  4653.8  244.64  4704.4  246.12  4833.6  243.98
  4890.8  243.05  4929.7   240.2  4970.8  235.31  4980.8  233.85    4997  229.16
  4999.8  228.66    5003  229.16  5020.8  235.51  5091.2  234.92  5180.8  238.14
  5270.8  238.76  5416.6  242.18    5525  247.27  5620.9  252.07  5650.9  255.21
  5790.9  265.33  5890.9  276.54    5911  282.08    5931     285  6147.7  293.49
#Mann= 8 ,-1 , 0
  3938.9     .05       0  4478.8      .1       0  4833.6     .05       0
  4929.7      .1       0    4997     .07       0    5003      .1       0
  5416.6     .05       0    5525      .1       0
Bank Sta=4970.8,5020.8
XS Rating Curve= 0 ,0
Exp/Cntr=0.3,0.1

Type RM Length L Ch R = 1 ,60530   ,1124,1124,1124
BEGIN DESCRIPTION:
SALT BRANCH 84.0
END DESCRIPTION:
XS GIS Cut Line= 3
      2220131.03     13312743.44      2222412.19     13312736.57
      2223043.54     13312448.35
#Sta/Elev= 30
    3077  263.99  3206.5  256.65  3363.7  245.87  3483.7  239.73  3563.7  236.87
  3649.2  237.06  3703.7  237.25  3743.7  232.23  3793.7  236.73  4016.6  235.84
  4233.7   234.3  4367.1  235.37  4523.7  237.01  4783.7  234.45  4873.7  235.38
  4963.7  234.44  4983.7  232.78  4993.7  229.97    4997   227.1  4999.8   226.6
    5003   227.1  5023.7  232.53  5043.7  234.09  5068.8  236.51  5293.7  248.73
  5438.7  249.73  5548.9  253.77  5639.5  257.21  5846.8   261.8  6052.2  270.88
#Mann= 9 ,-1 , 0
    3077      .1       0  3206.5     .05       0  3649.2      .1       0
  4016.6     .05       0  4367.1      .1       0    4997     .07       0
    5003      .1       0  5068.8     .05       0  5548.9      .1       0
#XS Ineff= 1 ,-1
 3702.54 3853.45  237.05
Permanent Ineff=
       F
Bank Sta=4963.7,5043.7
XS Rating Curve= 0 ,0
Exp/Cntr=0.3,0.1

Type RM Length L Ch R = 1 ,59406   ,365,365,365
BEGIN DESCRIPTION:
SALT BRANCH 83.0
END DESCRIPTION:
XS GIS Cut Line= 2
      2220330.35      13313437.4      2222623.92     13313183.32
#Sta/Elev= 30
    4075   269.4  4089.4  267.34  4132.7  261.41  4193.1  259.04  4323.9  250.38
  4484.2  243.39  4527.2  240.11  4645.8  232.36    4852  233.79  4947.7   232.4
  4987.9  229.34    4997  225.25  4999.8  224.75    5003  225.25    5008  225.25
  5018.1  229.76  5033.4  231.06    5169  234.16  5338.9  234.11  5682.1  236.58
  5758.9  236.06  5881.2  238.41  5945.3  239.61  5973.9  238.18    5994   239.8
  6074.5   241.5  6208.3  247.13  6245.6     248  6338.3  253.17  6382.6  254.88
#Mann= 9 ,-1 , 0
    4075      .1       0  4089.4     .05       0  4527.2      .1       0
    4997     .07       0    5003      .1       0  5338.9     .05       0
  5881.2      .1       0  6208.3     .05       0  6338.3      .1       0
#XS Ineff= 1 ,-1
 4600.64 4836.43  233.89
Permanent Ineff=
       F
Bank Sta=4987.9,5018.1
XS Rating Curve= 0 ,0
Exp/Cntr=0.3,0.1

Type RM Length L Ch R = 1 ,59041   ,533,533,533
BEGIN DESCRIPTION:
SALT BRANCH 82.0
END DESCRIPTION:
XS GIS Cut Line= 3
       2220772.4     13313784.36      2221172.44     13313734.35
      2222572.46     13313334.35
#Sta/Elev= 30
  4414.8  258.03  4435.1  257.88  4480.6  255.52  4611.6  254.71    4677  248.92
  4682.2  245.19  4692.3  242.34  4712.4  239.28  4722.5  238.91  4772.9  233.18
    4818  231.55  4833.8  229.87  4948.3  230.64  4958.7  230.15    4997  225.24
  4999.8  224.74    5003  225.24  5031.5  228.43  5073.1  230.49  5093.9  231.44
  5113.9  230.88  5197.9  232.32  5655.5  234.03  5863.5     237  5987.5   240.9
  6142.1  248.82  6165.1   250.6  6196.3  250.75  6237.9  254.58    6274  256.33
#Mann= 4 ,-1 , 0
  4414.8      .1       0    4997     .07       0    5003      .1       0
  6142.1     .05       0
#XS Ineff= 1 ,-1
 4790.89  4906.8   230.9
Permanent Ineff=
       F
Bank Sta=4948.3,5073.1
XS Rating Curve= 0 ,0
Exp/Cntr=0.3,0.1

Type RM Length L Ch R = 1 ,58508   ,844,844,844
BEGIN DESCRIPTION:
SALT BRANCH 81.0
END DESCRIPTION:
XS GIS Cut Line= 3
      2220962.48     13313918.37      2221477.76     13314117.61
      2222851.94     13313567.94
#Sta/Elev= 30
  4158.7  251.63    4199  251.57  4223.6  254.54  4283.4  250.76  4311.3  250.63
  4392.5  247.21  4417.1  247.55  4422.5  246.29  4441.7  247.14  4646.8  237.22
  4700.5  235.94  4770.7  237.15  4829.3  236.54  4834.7   235.1    4937  228.73
  4942.4  227.25    4972  226.24    4997  223.47  4999.8  222.97    5003  223.47
  5025.8  227.82  5128.2  227.39    5349  230.43  5432.7  230.08  5564.4  233.88
  5741.8  242.95  5833.6  247.83  5848.9  250.02  5941.3  256.24  6191.2  280.74
#Mann= 7 ,-1 , 0
  4158.7      .1       0  4311.3     .05       0  4770.7      .1       0
    4997     .07       0    5003      .1       0  5741.8     .08       0
  5848.9      .1       0
Bank Sta=4942.4,5025.8
XS Rating Curve= 0 ,0
Exp/Cntr=0.3,0.1

Type RM Length L Ch R = 1 ,57664   ,495,495,495
BEGIN DESCRIPTION:
SALT BRANCH 80.0
END DESCRIPTION:
XS GIS Cut Line= 3
      2221038.03     13314021.43      2221835.04     13314454.29
      2223202.35     13314413.06
#Sta/Elev= 30
  3501.6  246.66  3691.3  241.04  3777.5  237.03  3924.8  232.95  4006.5  233.27
    4170  238.74  4219.4  239.28  4251.7  241.24  4301.1  237.92  4362.5  235.82
  4407.2  233.04  4461.3  232.88  4641.4   228.8  4670.4  229.02  4721.4  229.55
  4911.5  225.16  4951.5  226.24  4991.5   224.1    4997  222.66  4999.8  222.16
    5003  222.66  5011.5  222.79  5021.5  225.64  5041.5   226.3  5085.9  226.24
  5184.2  231.11  5391.7  241.43  5601.8  253.76  5611.8  255.12  5776.5  263.91
#Mann= 9 ,-1 , 0
  3501.6      .1       0  3691.3     .05       0  4362.5      .1       0
  4461.3     .05       0  4670.4      .1       0    4997     .07       0
    5003      .1       0  5085.9     .05       0  5184.2      .1       0
Bank Sta=4951.5,5041.5
XS Rating Curve= 0 ,0
Exp/Cntr=0.3,0.1

Type RM Length L Ch R = 1 ,57169   ,773,773,773
BEGIN DESCRIPTION:
Mapping XS d2c02b58
END DESCRIPTION:
XS GIS Cut Line= 2
      2220928.12     13314990.21      2222858.81     13314859.67
#Sta/Elev= 30
  3622.1  253.99  3802.1  243.23  3912.4  238.03  3942.4  235.24  4033.3  232.84
  4099.3  229.83    4203  226.56  4453.6  225.54  4563.8  227.35  4864.5  224.86
  4924.7  223.31  4964.8  224.31  4984.8     222    4997     222  4999.8   221.5
    5003     222  5004.9  223.07  5014.9  223.66  5034.9  223.44  5044.9  224.43
    5075  226.54    5080  227.71  5095.1  227.45  5105.1  228.95  5196.1  233.66
  5294.8  239.62    5516  255.85  5536.1  257.74  5546.1  260.51  5557.2     262
#Mann= 7 ,-1 , 0
  3622.1      .1       0  4033.3     .05       0  4099.3      .1       0
    4997     .07       0    5003      .1       0  5196.1     .05       0
  5294.8      .1       0
Bank Sta=4964.8,5044.9
XS Rating Curve= 0 ,0
Exp/Cntr=0.3,0.1

Type RM Length L Ch R = 1 ,56396   ,487,487,487
BEGIN DESCRIPTION:
Mapping XS 8e695e64
END DESCRIPTION:
XS GIS Cut Line= 4
      2220632.67     13315608.59      2221175.44     13315505.53
      2222391.58     13315381.85      2222961.83     13314949.01
#Sta/Elev= 30
  3823.7  262.79  3971.7  262.68  4103.7  260.19  4185.8  255.31  4438.8  235.91
  4599.6  226.49  4760.4  221.43    4871  224.67  4951.4  223.76    4997  221.43
  4999.8  220.93    5003  221.43  5041.9  223.58    5072  222.47  5242.9  224.11
  5273.1  223.08  5293.2  225.22  5343.4  224.35  5716.9  230.69  5843.1  237.04
  6027.7  246.84  6056.8  249.42  6083.9  255.15    6113  257.31  6171.2  259.03
  6212.9  262.64    6242  261.95  6277.3  264.54  6291.9  264.02  6314.5  266.13
#Mann= 5 ,-1 , 0
  3823.7      .1       0    4997     .07       0    5003      .1       0
  5716.9     .05       0  5843.1      .1       0
Bank Sta=4951.4,5041.9
XS Rating Curve= 0 ,0
Exp/Cntr=0.3,0.1

Type RM Length L Ch R = 1 ,55909   ,553,553,553
BEGIN DESCRIPTION:
SALT BRANCH 77.0
END DESCRIPTION:
XS GIS Cut Line= 3
      2220790.65      13316316.3      2221312.86     13316117.04
       2223236.7     13315079.53
#Sta/Elev= 30
    3944  269.72  4181.3  261.46  4502.9  246.35  4552.1  244.83  4636.5  245.11
  4640.2     245  4743.5   241.5  4749.2  239.94  4787.3  239.77  4792.9   237.7
  4825.4  235.22  4831.1  232.39  4874.8  226.38  4928.8  223.04    4997  220.49
  4999.8  219.99    5003  220.49  5053.8  223.13  5082.4  222.18  5201.5  223.21
  5246.2  222.81  5328.1  224.35  5339.5  225.36  5383.3  223.65  5487.1  222.94
  5829.6  227.02    5943  228.73  6071.8  231.98  6410.7  246.79  6688.7  255.61
#Mann= 9 ,-1 , 0
    3944      .1       0  4636.5     .05       0  4640.2      .1       0
    4997     .07       0    5003      .1       0  5201.5     .16       0
  5328.1      .1       0  5829.6     .05       0    5943      .1       0
Bank Sta=4928.8,5053.8
XS Rating Curve= 0 ,0
Exp/Cntr=0.3,0.1

Type RM Length L Ch R = 1 ,55356   ,224,224,224
BEGIN DESCRIPTION:
Mapping XS 2fbdb859
END DESCRIPTION:
XS GIS Cut Line= 3
      2220735.06     13316836.87      2222071.89     13316333.39
      2223399.99     13315526.12
#Sta/Elev= 30
  3627.4  253.53    3772  253.09  3878.1   252.5  4047.3  246.44  4196.5  241.86
  4271.3  240.06    4505  234.73  4669.9  238.09  4772.4  241.15  4863.1  232.17
    4943  219.19  4972.4  219.23  4987.3  219.23    4997  216.53  4999.8  216.03
    5003  216.53  5003.4  219.31  5045.7  219.24  5086.1  228.24  5129.9  221.83
  5161.7  221.36    5364  221.46  5391.2  216.53    5428  221.45  5512.8  221.86
  5629.9  220.73  5997.6  221.62  6317.4  231.79  6432.1   237.1  6610.1   248.4
#Mann= 18 ,-1 , 0
  3627.4      .1       0    3772     .08       0  3878.1     .05       0
  4047.3      .1       0  4196.5     .05       0  4271.3      .1       0
    4505     .05       0  4669.9      .1       0  4972.4     .05       0
    4997    .033       0    5003     .05       0  5045.7      .1       0
  5129.9     .16       0  5161.7      .1       0  5512.8     .05       0
  5629.9      .1       0  6317.4     .05       0  6432.1      .1       0
Bank Sta=4987.3,5003.4
XS Rating Curve= 0 ,0
Exp/Cntr=0.3,0.1

Type RM Length L Ch R = 1 ,55132   ,445,445,445
BEGIN DESCRIPTION:
SALT BRANCH 76.0
END DESCRIPTION:
XS GIS Cut Line= 3
      2220819.24      13317078.2       2222204.7     13316505.27
      2223631.82     13315656.29
#Sta/Elev= 30
  3575.2  241.11  3889.5  235.94  4106.5  233.32  4590.1  229.32    4619  229.71
  4822.6  235.41  4991.1  226.34    4997  214.64  4999.8  214.14    5003  214.64
  5006.1  226.91  5020.5  226.52  5063.3  226.71  5103.9  226.59  5119.5  221.01
  5125.3  222.98  5156.5  217.57  5279.1  221.94  5365.2  220.97  5481.5  217.99
    5507  214.67  5555.7  220.66  5592.7  218.16  5608.3  220.32  5629.7  216.29
  5645.3  219.82    5842   217.7  6095.7  223.12  6427.8  240.11    6735  263.54
#Mann= 13 ,-1 , 0
  3575.2      .1       0  3889.5     .05       0  4106.5      .1       0
  4590.1     .05       0    4619      .1       0    4997     .07       0
    5003      .1       0  5020.5     .05       0  5063.3      .1       0
  5365.2     .05       0  5481.5      .1       0  6095.7     .05       0
  6427.8      .1       0
Bank Sta=4991.1,5006.1
XS Rating Curve= 0 ,0
Exp/Cntr=0.3,0.1

Type RM Length L Ch R = 1 ,54687   ,402,402,402
BEGIN DESCRIPTION:
SALT BRANCH 75.0
END DESCRIPTION:
XS GIS Cut Line= 2
      2221134.19     13317333.19      2223786.11     13315821.74
#Sta/Elev= 30
  3478.8  243.05  4051.9  228.63  4150.1  227.08  4391.8  224.42  4415.7  224.44
  4980.4  217.59  4990.7  214.23    4997  213.94  4999.8  213.44    5003  213.94
  5017.9   218.3  5039.5  220.46    5077  217.41  5105.7  220.75  5238.3  219.92
  5244.1  216.66  5259.9  215.85  5281.5  218.13    5319  215.87  5324.7  219.44
  5334.8  219.78  5393.6  214.22  5442.9  219.77  5508.7  214.85  5531.7  218.51
  5625.8   216.6  6072.7  237.28  6330.3  256.82  6454.2  274.14  6531.2  275.88
#Mann= 9 ,-1 , 0
  3478.8      .1       0  4051.9     .05       0  4150.1      .1       0
  4391.8     .05       0  4415.7      .1       0  4990.7     .05       0
    4997     .04       0    5003     .05       0  5105.7      .1       0
Bank Sta=4980.4,5017.9
XS Rating Curve= 0 ,0
Exp/Cntr=0.3,0.1

Type RM Length L Ch R = 1 ,54285   ,736,736,736
BEGIN DESCRIPTION:
SALT BRANCH 74.0
END DESCRIPTION:
XS GIS Cut Line= 2
      2221388.46     13317532.42       2223779.5       13316385.
#Sta/Elev= 30
  3573.3  243.04    3750  235.56  3870.8  232.65  3957.2   232.2  4017.7  231.87
  4080.1  226.87  4146.9  223.69  4266.9  221.04  4644.2  219.59  4881.3   220.1
    4921  218.59  4934.8  217.39  4980.1  215.33    4997  211.56  4999.8  211.06
    5003  211.56  5036.6  217.24  5098.9  219.98  5285.6  218.69  5369.4  216.66
  5376.2  214.82  5413.7   214.6  5421.5  211.56  5449.7  215.62  5466.8  215.97
  5489.4  218.79  5681.7  226.07  5979.2  241.65  6119.3  249.99  6225.4  257.65
#Mann= 9 ,-1 , 0
  3573.3      .1       0  3957.2     .05       0  4146.9      .1       0
  4644.2     .05       0    4921      .1       0    4997     .07       0
    5003      .1       0  5979.2     .05       0  6119.3      .1       0
Bank Sta=4934.8,5036.6
XS Rating Curve= 0 ,0
Exp/Cntr=0.3,0.1

Type RM Length L Ch R = 1 ,53549   ,531,531,531
BEGIN DESCRIPTION:
SALT BRANCH 73.0
END DESCRIPTION:
XS GIS Cut Line= 3
      2221687.69     13317896.87      2223287.72     13317246.85
      2223637.69     13317046.87
#Sta/Elev= 30
  3245.3  237.96    3493   225.2  3522.4  222.69  3546.5  222.68  3644.7  219.06
  3707.2  217.61    3742  218.25  3784.8  217.39  4088.2  217.36  4189.2   217.9
  4320.3  216.58  4588.1  218.66  4646.9  217.84  4842.8  218.34  4928.1  215.18
  4957.6  212.16  4980.2  213.12    4986  212.77  4995.4  210.21    4997  208.98
  4999.8  208.48    5003  208.98  5007.6  209.41  5017.7  213.91  5023.4  217.85
  5039.3  221.23    5076  224.77  5104.1  226.28  5119.9  228.32  5375.4  241.92
#Mann= 5 ,-1 , 0
  3245.3      .1       0  4088.2     .05       0  4646.9      .1       0
    4997     .07       0    5003      .1       0
Bank Sta=4980.2,5017.7
XS Rating Curve= 0 ,0
Exp/Cntr=0.3,0.1

Type RM Length L Ch R = 1 ,53018   ,693,693,693
BEGIN DESCRIPTION:
SALT BRANCH 72.0
END DESCRIPTION:
XS GIS Cut Line= 3
      2221737.73     13319296.85      2223337.72     13317746.85
      2223837.73     13317146.84
#Sta/Elev= 30
  2773.7  249.51  2985.8  241.72  3254.6  234.36  3530.4  235.92  3644.3  231.31
  3671.8  228.12  3827.5  220.97  4151.9  215.81  4379.5  214.78  4497.5  215.12
  4635.1  214.92  4767.1  215.63  4909.4  214.61  4930.7  212.41  4937.7  213.71
  4980.1  212.83  4987.3  208.34    4997  207.53  4999.8  207.03    5003  207.53
  5008.5  207.53    5015  209.87  5022.8  209.58  5029.3  212.81  5051.5   213.6
    5058  215.51  5378.2  224.83    5399  227.57  5626.2     239  5782.4   249.7
#Mann= 9 ,-1 , 0
  2773.7      .1       0  3644.3     .05       0  4151.9      .1       0
  4379.5     .05       0  4497.5      .1       0  4635.1     .05       0
  4767.1      .1       0    4997     .07       0    5003      .1       0
Bank Sta=4980.1,5029.3
XS Rating Curve= 0 ,0
Exp/Cntr=0.3,0.1

Type RM Length L Ch R = 1 ,52325   ,843,843,843
BEGIN DESCRIPTION:
SALT BRANCH 71.0
END DESCRIPTION:
XS GIS Cut Line= 3
      2223058.06     13319662.38      2223161.12     13318982.19
      2224033.72     13317230.12
#Sta/Elev= 30
  3677.7  246.33  3841.2  238.43  4042.5  231.22  4360.8  222.97  4588.8  215.29
  4703.5  212.32  4740.3  208.98  4748.2  211.97  4762.6  211.77  4770.6  213.36
  4874.3  214.16  4955.3  212.99  4963.7  211.46  4972.1  212.38  4977.7   208.8
    4997  206.96  4999.8  206.46    5003  206.96  5016.9  207.29  5022.5   211.4
  5030.7  209.02  5039.3   208.7  5067.2  212.73  5151.2   215.3  5554.2  213.78
  5611.7  215.08  6046.7  235.24  6184.6  244.18  6248.2  249.22    6323  251.92
#Mann= 5 ,-1 , 0
  3677.7     .05       0  4588.8      .1       0    4997     .07       0
    5003      .1       0  6184.6     .05       0
Bank Sta=4972.1,5022.5
XS Rating Curve= 0 ,0
Exp/Cntr=0.3,0.1

Type RM Length L Ch R = 1 ,51482   ,528,528,528
BEGIN DESCRIPTION:
SALT BRANCH 70.0
END DESCRIPTION:
XS GIS Cut Line= 3
      2224088.68     13319524.98       2224061.2     13318920.35
      2224095.56     13317484.32
#Sta/Elev= 30
  4240.6  236.14    4509  226.31    4539  226.42  4769.3     218  4819.3  217.22
  4829.3   218.1  4839.3  215.42  4948.6  211.61  4969.4  210.43  4990.9  207.34
    4997     205  4999.8   204.5    5003     205  5029.4  210.51  5089.4  210.29
  5159.4  213.04  5239.5  211.01    5331  212.91  5439.5  211.99  5469.5  212.59
  5629.6  210.77  5709.6  212.46  5869.6  219.54  5879.6  220.76  5919.7  220.73
  5959.7  222.23  5989.7  225.49  6019.7  226.39  6069.7  230.52  6282.3  242.29
#Mann= 5 ,-1 , 0
  4240.6      .1       0  4948.6     .07       0  4990.9      .1       0
    4997     .07       0    5003      .1       0
Bank Sta=4969.4,5029.4
XS Rating Curve= 0 ,0
Exp/Cntr=0.3,0.1

Type RM Length L Ch R = 1 ,50954   ,729,729,729
BEGIN DESCRIPTION:
SALT BRANCH 69.0
END DESCRIPTION:
XS GIS Cut Line= 3
      2224624.61     13319394.48      2224535.29     13317841.62
      2224287.92      13317463.7
#Sta/Elev= 30
    4314  242.81  4351.8  239.36  4451.8  234.21    4519  229.42    4524  230.36
    4572  226.74  4622.1  225.18  4696.2   220.6  4892.6  212.29  4922.6  207.84
  4952.7  206.66  4962.7  207.71  4972.7  205.66  4982.7   205.8  4992.7  202.51
    4997  202.51  4999.8  202.01    5003  202.51  5012.8  208.22  5032.8  211.07
  5082.9  211.38    5163  209.71  5243.2  210.66  5583.7  209.69    5774  216.45
    5784  217.83  5844.1  219.66  6073.6  232.03  6253.6   239.9  6321.1  241.69
#Mann= 4 ,-1 , 0
    4314      .1       0    4997     .07       0    5003      .1       0
  6253.6     .05       0
Bank Sta=4962.7,5012.8
XS Rating Curve= 0 ,0
Exp/Cntr=0.3,0.1

Type RM Length L Ch R = 1 ,50225   ,611,611,611
BEGIN DESCRIPTION:
SALT BRANCH 68.0
END DESCRIPTION:
XS GIS Cut Line= 3
      2225318.57     13319236.42      2225057.48     13317731.69
       2224342.9     13317346.92
#Sta/Elev= 30
  4289.3  231.82  4481.7   223.8  4522.3  220.97  4684.7     215  4806.5  212.09
  4836.9  210.33  4948.6   208.5    4979  205.86  4989.2  203.92    4997  200.63
  4999.8  200.13    5003  200.63  5009.5  204.38  5025.1  209.34    5182  209.23
  5258.8  207.79  5313.4  208.39  5334.3  206.29  5354.6  208.31  5537.2  210.86
  5816.4  214.13    5961  214.64  6196.3  221.88    6322  227.18  6409.6  229.19
  6469.7  232.43  6507.8  233.24  6513.5  232.46  6573.5  235.85  6628.1  237.43
#Mann= 3 ,-1 , 0
  4289.3      .1       0    4997     .07       0    5003      .1       0
Bank Sta=4948.6,5025.1
XS Rating Curve= 0 ,0
Exp/Cntr=0.3,0.1

Type RM Length L Ch R = 1 ,49614   ,576,576,576
BEGIN DESCRIPTION:
SALT BRANCH 67.0
END DESCRIPTION:
XS GIS Cut Line= 2
      2225675.85     13318975.36      2225950.69     13317175.12
#Sta/Elev= 30
    4400  232.51  4459.2   233.2  4540.1  230.23  4661.5  224.24  4782.9  215.62
  4904.3  209.41  4909.3  208.01  4954.9  206.31  4977.9  206.72  4985.2  205.09
    4997  198.36  4999.8  197.86    5003  198.36  5005.4  198.36  5015.6  204.25
  5025.7  205.82  5082.7  206.67  5136.9  206.06  5167.3  203.03  5191.7  204.98
  5241.9  206.43  5329.1  206.27  5410.1   208.4  5683.2  219.12  5895.6  232.25
  5946.2  235.92  5956.3   237.9  5970.5  238.18  5996.8  241.34  6221.1  254.73
#Mann= 5 ,-1 , 0
    4400      .1       0    4997     .07       0    5003      .1       0
  5082.7     .12       0  5191.7      .1       0
Bank Sta=4977.9,5025.7
XS Rating Curve= 0 ,0
Exp/Cntr=0.3,0.1

Type RM Length L Ch R = 1 ,49038   ,1288,1288,1288
BEGIN DESCRIPTION:
SALT BRANCH 66.0
END DESCRIPTION:
XS GIS Cut Line= 4
       2225469.7     13319208.94      2226156.81     13318892.86
      2226651.52     13317628.63       2226432.2     13317176.29
#Sta/Elev= 30
  3852.5     231  3971.4  231.91  4057.4  229.26  4062.9  229.98  4213.6  225.93
  4321.1  221.66  4372.6  221.27  4395.5  219.43  4515.9  216.39  4532.8  214.69
  4606.6  212.04  4677.1  211.99  4797.8  207.93  4978.4  204.18  4983.8   203.5
    4997  198.36  4999.8  197.86    5003  198.36  5023.3  203.38  5032.7  203.79
  5152.2  205.91  5260.6  204.65  5399.2  205.18  5724.7  209.72  5936.1  213.94
  5964.7  215.52  6068.4   216.2  6279.3  225.91  6290.7  227.73  6469.1  237.69
#Mann= 3 ,-1 , 0
  3852.5      .1       0    4997     .07       0    5003      .1       0
Bank Sta=4978.4,5032.7
XS Rating Curve= 0 ,0
Exp/Cntr=0.3,0.1

Type RM Length L Ch R = 1 ,47750   ,688,688,688
BEGIN DESCRIPTION:
SALT BRANCH 65.0
END DESCRIPTION:
XS GIS Cut Line= 2
       2225490.3     13319270.77      2227604.68     13318749.04
#Sta/Elev= 30
  3631.6  231.82  3639.2  232.47    3755  230.41  3855.5  226.73  3879.4  226.62
  3915.7  224.47  3998.7  222.86  4102.7  218.68    4113  217.39  4123.1  217.69
  4169.7  214.75  4335.6  207.16    4460  203.63  4576.5  204.31  4874.7  203.91
  4957.6  202.54  4978.2   201.2  4988.5   197.1    4997  194.94  4999.8  194.44
    5003  194.94  5029.7  199.98  5050.9  199.97  5122.4   203.4  5175.3  207.52
  5318.1  216.17  5507.1  225.84  5699.2  238.14  5797.4  246.11  5809.4   246.4
#Mann= 3 ,-1 , 0
  3631.6      .1       0    4997     .07       0    5003      .1       0
Bank Sta=4978.2,5029.7
XS Rating Curve= 0 ,0
Exp/Cntr=0.3,0.1

Type RM Length L Ch R = 1 ,47062   ,1239,1239,1239
BEGIN DESCRIPTION:
SALT BRANCH 64.0
END DESCRIPTION:
XS GIS Cut Line= 3
      2225181.16     13319882.27       2227338.6     13319531.85
        2227689.     13318995.95
#Sta/Elev= 30
  3149.9  237.71  3409.8  228.08  3480.7  226.52  3490.9  225.29    3886  214.93
  3962.7  213.64  4090.9  216.05  4189.9  212.22  4281.1  205.63  4362.1  202.37
  4453.3  201.28  4574.9  202.66  4583.5  201.69  4655.9  200.91  4696.5  199.22
  4834.9  199.59  4868.7  200.74    4970  198.56  4990.3  194.11    4997  191.65
  4999.8  191.15    5003  191.65  5010.5  195.89  5019.7  198.46  5024.7   197.7
  5091.6  200.63  5339.4  201.84  5438.8  205.75  5728.4   223.1  5975.9  244.43
#Mann= 3 ,-1 , 0
  3149.9      .1       0    4997     .07       0    5003      .1       0
Bank Sta=4970,5019.7
XS Rating Curve= 0 ,0
Exp/Cntr=0.3,0.1

Type RM Length L Ch R = 1 ,45823   ,843,843,843
BEGIN DESCRIPTION:
SALT BRANCH 62.0
END DESCRIPTION:
XS GIS Cut Line= 3
      2225682.73     13321483.18      2226569.07     13321311.41
      2227771.49     13319126.44
#Sta/Elev= 30
  3042.2  224.66    3413  209.92  3607.5  206.61  3719.6  206.77  3801.1  209.89
  3882.5  215.19  3948.8  216.94  4242.1  203.73  4388.9  199.51  4454.3  200.61
  4650.8  210.52  4807.5  218.02    4852  215.68  4874.8  212.71  4883.2  210.15
  4911.2  207.24  4942.9  199.33  4977.5  195.49  4986.4  190.59  4992.2  191.35
    4997  186.76  4999.8  186.26    5003  186.76  5008.2  193.12  5023.2  195.05
  5251.4  199.28  5861.5  200.32    5959   203.9  6089.7  211.39    6439  237.99
#Mann= 5 ,-1 , 0
  3042.2      .1       0  4650.8     .05       0  4911.2      .1       0
    4997     .07       0    5003      .1       0
Bank Sta=4977.5,5023.2
XS Rating Curve= 0 ,0
Exp/Cntr=0.3,0.1

Type RM Length L Ch R = 1 ,44980   ,1086,1086,1086
BEGIN DESCRIPTION:
SALT BRANCH 61.0
END DESCRIPTION:
XS GIS Cut Line= 4
      2227695.89      13322115.3      2227888.27     13321764.89
      2227936.37     13318940.96      2227936.37     13318968.48
#Sta/Elev= 30
  3325.9  222.13  3384.3  219.96  3487.5  214.14  3540.9  209.56  3597.9  207.46
  3656.2  201.41  3672.3  200.61  3694.1  201.85  3773.7   197.2  3933.7  191.88
  3982.8  194.54  4571.4  194.03  4783.8  196.29  4973.9  193.17  4983.9  188.94
    4997  187.09  4999.8  186.59    5003  187.09  5013.9  193.13  5193.9  196.39
  5463.9  195.98  5743.8  200.39    5924  209.18    6024  215.05    6134  223.39
    6214  227.29    6244  230.67  6504.1  250.41  6544.1  252.28  6577.5   251.6
#Mann= 3 ,-1 , 0
  3325.9      .1       0    4997     .07       0    5003      .1       0
Bank Sta=4973.9,5013.9
XS Rating Curve= 0 ,0
Exp/Cntr=0.3,0.1

Type RM Length L Ch R = 1 ,43894   ,589,589,589
BEGIN DESCRIPTION:
SALT BRANCH 59.0
END DESCRIPTION:
XS GIS Cut Line= 3
       2227487.7     13322446.88      2228637.72     13321196.85
      2229887.73     13319746.84
#Sta/Elev= 30
  3318.6  245.42  3346.7  245.37  3382.4  240.54  3502.7  233.04  3757.3  224.49
  3870.7  216.43  3905.9  216.22    3991  211.18  4019.3  207.99  4309.7  193.82
  4436.7  190.72  4444.1   188.5  4493.4  187.95  4521.8  191.62  4564.3  192.36
  4960.7  189.98  4989.1  187.86    4997  182.61  4999.8  182.11    5003  182.61
  5030.9  190.09  5087.9  192.47  5364.4  191.72  5605.7  197.53  5832.8  196.77
  5939.3   199.7  6137.8  209.49  6428.6  228.45  6449.4  228.29  6931.6  262.69
#Mann= 3 ,-1 , 0
  3318.6      .1       0    4997     .07       0    5003      .1       0
Bank Sta=4960.7,5030.9
XS Rating Curve= 0 ,0
Exp/Cntr=0.3,0.1

Type RM Length L Ch R = 1 ,43305   ,1041,1041,1041
BEGIN DESCRIPTION:
SALT BRANCH 58.0
END DESCRIPTION:
XS GIS Cut Line= 3
      2228156.25      13322603.1      2228417.33     13321971.01
      2229729.25     13320281.31
#Sta/Elev= 30
  4067.1  239.74  4109.6  237.98  4377.2  222.24  4472.9  215.16  4478.3  215.78
  4608.7  208.81  4715.2   202.8  4750.5  199.75  4796.5  198.68    4811  196.96
  4968.4  189.88  4974.8  187.34    4997  182.11  4999.8  181.61    5003  182.11
  5010.1  184.96  5053.5  189.27  5082.5  189.27  5110.7  191.18    5288  192.33
  5652.7  191.29  5731.1  190.03  5866.3  192.79  6059.1  191.34  6300.8  194.15
  6436.5  199.15  6579.3  207.14  6793.1  221.23  6849.2  223.84  6890.2  227.62
#Mann= 4 ,-1 , 0
  4067.1     .05       0  4109.6      .1       0    4997     .07       0
    5003      .1       0
Bank Sta=4968.4,5053.5
XS Rating Curve= 0 ,0
Exp/Cntr=0.3,0.1

Type RM Length L Ch R = 1 ,42264   ,654,654,654
BEGIN DESCRIPTION:
SALT BRANCH 57.0
END DESCRIPTION:
XS GIS Cut Line= 3
      2228382.95     13322857.37      2229111.29     13322362.65
      2230112.95     13320462.24
#Sta/Elev= 30
  3833.9  230.79  3952.5  235.36  4060.3  233.39  4377.6   216.4  4541.6  210.59
  4710.7  197.76  4782.4  193.49  4958.7  189.04    4975  186.14  4980.9  181.32
    4997  177.46  4999.8  176.96    5003  177.46  5003.5  180.71  5013.4  184.84
  5041.1  184.34  5079.5  188.42  5426.3  189.38  5580.5  188.29  5596.9  185.94
  5625.2  185.82  5679.3  189.88    5685  192.35  5849.9  190.78  6086.5  198.86
  6279.1   200.3  6515.8  212.66  6603.9  220.07  6664.3  222.65  6862.6  239.49
#Mann= 5 ,-1 , 0
  3833.9      .1       0  4541.6     .05       0  4710.7      .1       0
    4997     .07       0    5003      .1       0
Bank Sta=4975,5013.4
XS Rating Curve= 0 ,0
Exp/Cntr=0.3,0.1

Type RM Length L Ch R = 1 ,41610   ,520,520,520
BEGIN DESCRIPTION:
SALT BRANCH 55.0
END DESCRIPTION:
XS GIS Cut Line= 3
      2229640.34     13323235.25      2229736.53     13322383.26
      2230547.32     13320892.25
#Sta/Elev= 30
  3838.7   208.3  4022.1  203.08  4130.8   199.7  4219.3  197.56  4425.8  195.84
  4664.7  191.83  4834.5  186.97  4921.9  186.77  4953.8  184.15  4965.6   183.7
    4997  178.45  4999.8  177.95    5003  178.45  5010.7  179.68  5019.7   183.6
    5079     186  5608.7  187.04  5734.1  193.85  5784.8  199.09  5875.7  205.65
  5887.2  207.96  5919.4  209.29  5968.8  215.06  6088.5  224.67  6094.2  226.32
  6132.2  228.05  6154.1   230.5  6257.6  234.91  6263.3  236.55  6393.3  240.08
#Mann= 7 ,-1 , 0
  3838.7      .1       0  4022.1     .05       0  4130.8      .1       0
  4219.3     .05       0  4425.8      .1       0    4997     .07       0
    5003      .1       0
Bank Sta=4953.8,5019.7
XS Rating Curve= 0 ,0
Exp/Cntr=0.3,0.1

Type RM Length L Ch R = 1 ,41090   ,795,795,795
BEGIN DESCRIPTION:
SALT BRANCH 54.0
END DESCRIPTION:
XS GIS Cut Line= 3
       2229687.7     13323646.89      2230387.72     13322096.85
      2230687.74     13321396.81
#Sta/Elev= 30
  3283.8  222.79  3534.8  212.19  3563.4  212.37    3592  209.97  3736.3  203.86
  4024.7  194.29  4168.9  192.19  4205.5  192.73  4468.9  188.27  4583.9  188.14
  4733.6  184.77  4854.7  185.12  4940.7  183.52  4970.3  181.53  4975.8  179.41
  4987.3   179.3    4997  177.62  4999.8  177.12    5003  177.62  5017.2  179.71
  5028.1  184.98  5191.3  184.46  5321.8  189.91  5495.9  202.71  5532.2  207.11
  5561.2   213.1  5593.8  215.26  5702.6  226.96  5713.5  229.51  5746.2  231.74
#Mann= 3 ,-1 , 0
  3283.8      .1       0    4997     .07       0    5003      .1       0
Bank Sta=4940.7,5028.1
XS Rating Curve= 0 ,0
Exp/Cntr=0.3,0.1

Type RM Length L Ch R = 1 ,40295   ,1073,1073,1073
BEGIN DESCRIPTION:
Mapping XS 3f760ebf
END DESCRIPTION:
XS GIS Cut Line= 3
      2230564.89     13323672.39      2230912.12     13323030.02
      2230946.84     13321363.39
#Sta/Elev= 30
  3852.7  207.42  3869.5  206.45  3998.2  200.13    4140  196.18  4249.4  195.47
  4331.3  197.68  4369.4  196.42  4413.1  197.07  4534.4  189.96  4544.2   189.9
  4771.3  187.87    4915  186.53  4966.2  185.28  4976.2   180.4    4997  176.32
  4999.8  175.82    5003  176.32  5016.2  180.79  5036.2  181.92  5106.2  180.96
  5146.2  182.92  5166.2  181.86  5266.2  183.41  5546.3  182.14  5656.3   183.6
  5736.3  188.37  5876.4  201.65  5976.4  208.81  6066.4  213.06  6249.9  217.58
#Mann= 8 ,-1 , 0
  3852.7     .05       0  3869.5      .1       0  4534.4     .05       0
  4544.2      .1       0  4771.3     .05       0    4915      .1       0
    4997     .07       0    5003      .1       0
Bank Sta=4976.2,5016.2
XS Rating Curve= 0 ,0
Exp/Cntr=0.3,0.1

Type RM Length L Ch R = 1 ,39222   ,924,924,924
BEGIN DESCRIPTION:
SALT BRANCH 52.0
END DESCRIPTION:
XS GIS Cut Line= 4
      2232153.45     13324002.27      2231806.22     13323264.39
      2231684.69     13321198.42       2231545.8     13320773.07
#Sta/Elev= 30
  3205.7  218.63  3266.9  215.83  3275.2  213.65  3280.7  215.11    3298  211.98
  3320.8  213.17  3326.3  210.81  3394.7  211.33    3776  195.63    4179  183.64
  4449.5  180.83  4659.8  180.98  4689.9  182.06  4900.3  178.63  4950.3  179.58
    4997  173.56  4999.8  173.06    5003  173.56  5020.5  177.16  5040.5  176.94
  5070.5  179.59  5090.6  179.02    5104  180.88  5160.7  183.56  5200.8   183.5
    5321  187.99  5461.2   189.6  5571.4  188.44  5831.9  191.68  6538.2  214.75
#Mann= 3 ,-1 , 0
  3205.7      .1       0    4997     .07       0    5003      .1       0
Bank Sta=4950.3,5070.5
XS Rating Curve= 0 ,0
Exp/Cntr=0.3,0.1

Type RM Length L Ch R = 1 ,38298   ,539,539,539
BEGIN DESCRIPTION:
Mapping XS dda8e61b
END DESCRIPTION:
XS GIS Cut Line= 2
      2232932.12     13323480.95      2232142.52     13321372.45
#Sta/Elev= 30
  4028.1  243.01    4082  235.39  4106.9  232.58  4112.3  233.05  4137.2  228.54
  4172.8  225.88  4252.9  215.87  4523.7  192.41  4625.2  185.83  4765.9  179.76
  4856.7     177  4942.2  176.05  4967.1  177.27  4982.8  175.53    4992  169.85
    4997  169.36  4999.8  168.86    5003  169.36  5022.3  175.14  5052.6  178.19
  5077.5  177.22  5138.1   177.9  5193.3  180.44  5312.1  182.99  5455.1  182.61
  5565.5   186.8  5741.8  188.06  5770.9  189.97  5852.2  188.75  6279.6  193.05
#Mann= 5 ,-1 , 0
  4028.1      .1       0    4997     .07       0    5003      .1       0
  5312.1     .05       0  5770.9      .1       0
Bank Sta=4982.8,5022.3
XS Rating Curve= 0 ,0
Exp/Cntr=0.3,0.1

Type RM Length L Ch R = 1 ,37759   ,492,492,492
BEGIN DESCRIPTION:
Mapping XS bab9723a
END DESCRIPTION:
XS GIS Cut Line= 2
      2233279.36     13322934.11      2232558.86     13321215.32
#Sta/Elev= 30
  4230.4  194.16  4298.6  188.36  4411.8  181.33  4563.6  176.12  4650.3  175.51
  4726.2  176.62  4812.1  174.43  4894.3  176.11  4947.2  176.25  4976.4  174.29
  4994.8  171.67    4997  168.67  4999.8  168.17    5003  168.67  5008.1  170.66
  5029.8  175.45  5053.2  176.61  5094.9  176.96  5159.9  182.12  5204.8  182.76
  5317.4  183.62  5403.6  183.95  5436.9   183.3  5518.9  183.94    5702  190.09
  5864.8  197.25  5940.6  201.25  6032.6  202.29  6056.4  204.01  6094.1  204.82
#Mann= 9 ,-1 , 0
  4230.4      .1       0    4997     .07       0    5003      .1       0
  5204.8     .05       0  5317.4      .1       0  5403.6     .05       0
  5518.9      .1       0    5702     .05       0  5864.8      .1       0
Bank Sta=4947.2,5029.8
XS Rating Curve= 0 ,0
Exp/Cntr=0.3,0.1

Type RM Length L Ch R = 1 ,37267   ,541,541,541
BEGIN DESCRIPTION:
SALT BRANCH 48.0
END DESCRIPTION:
XS GIS Cut Line= 3
      2233787.73     13322746.88      2233387.72     13321946.85
      2232837.71     13321146.84
#Sta/Elev= 30
  4120.3  216.28    4179  205.67  4285.2  193.63  4402.6  185.11  4478.1  176.29
  4537.8  173.96  4693.3  175.33  4805.1  174.87  4858.2  173.04    4970  174.25
    4984   172.4    4997  167.78  4999.8  167.28    5003  167.78  5006.4  167.78
    5012  172.07  5017.8  172.07  5022.2  174.39  5043.2  175.68  5093.9  174.82
  5167.2  177.83  5190.6  178.46  5309.5  184.24  5380.7  186.95  5467.3  185.98
  5560.8  187.71  5691.3     195  5796.1  198.55  5891.5  204.88  5985.6  213.95
#Mann= 8 ,-1 , 0
  4120.3     .05       0  4537.8      .1       0    4997     .07       0
    5003      .1       0  5167.2     .05       0  5190.6      .1       0
  5309.5     .05       0  5796.1      .1       0
Bank Sta=4970,5022.2
XS Rating Curve= 0 ,0
Exp/Cntr=0.3,0.1

Type RM Length L Ch R = 1 ,36726   ,378,378,378
BEGIN DESCRIPTION:
SALT BRANCH 47.0
END DESCRIPTION:
XS GIS Cut Line= 3
      2234037.72     13322546.87      2233937.72     13321896.85
       2233337.7     13321096.83
#Sta/Elev= 30
  4309.7  205.35  4350.2  203.75  4379.3   200.9  4479.7   190.5    4580  182.94
  4680.4  175.61  4754.9  172.71  4974.7  172.45  4995.5  169.54    4997  166.83
  4999.8  166.33    5003  166.83  5024.7  173.76  5060.1  172.81  5103.8  173.93
  5174.7  173.88  5210.1  175.31  5217.4  174.35  5374.7  173.79  5460.1  177.86
  5653.8  180.07  5674.7  180.92  5689.2  182.72  5710.1  183.14  5739.2  186.39
  5760.1  186.23    5821  189.81  5895.5  195.08  5930.9  199.52  5967.4  201.31
#Mann= 8 ,-1 , 0
  4309.7      .1       0  4379.3     .05       0  4479.7      .1       0
    4580     .05       0  4680.4      .1       0    4997     .07       0
    5003      .1       0    5821     .05       0
Bank Sta=4974.7,5024.7
XS Rating Curve= 0 ,0
Exp/Cntr=0.3,0.1

Type RM Length L Ch R = 1 ,36348   ,752,752,752
BEGIN DESCRIPTION:
SALT BRANCH 46.0
END DESCRIPTION:
XS GIS Cut Line= 3
      2234314.91     13322743.53      2234497.19     13322179.32
       2233750.7     13320781.83
#Sta/Elev= 30
  3944.5  190.74  4350.9  182.27  4536.1  176.55  4634.2  176.75  4665.6  175.64
  4793.4  172.98  4902.5  170.68    4974  172.07  4982.4  170.55  4990.3  166.52
    4997  166.52  4999.8  166.02    5003  166.52  5012.3  172.06  5078.1   173.8
  5204.2  172.01  5357.8  173.56  5626.1  173.44  5675.7  174.35    5818  181.31
  5883.9  181.68  5905.8   183.5  5934.7  183.43  6053.8  187.51  6075.7  186.67
    6092  188.13  6097.7   187.2    6114  188.51  6119.6  187.87  6121.8  188.94
#Mann= 5 ,-1 , 0
  3944.5      .1       0  4665.6     .05       0  4793.4      .1       0
    4997     .07       0    5003      .1       0
Bank Sta=4974,5012.3
XS Rating Curve= 0 ,0
Exp/Cntr=0.3,0.1

Type RM Length L Ch R = 1 ,35596   ,679,679,679
BEGIN DESCRIPTION:
Mapping XS ccd08557
END DESCRIPTION:
XS GIS Cut Line= 3
      2235282.25     13322480.76      2235146.72     13321791.81
      2233785.85     13320052.61
#Sta/Elev= 30
  3891.5  187.54  3956.6  187.13    4049  183.61  4171.7  181.43  4293.2  179.48
  4415.3  177.37  4466.2  178.26  4527.4  175.68  4557.7  176.25  4603.2  174.38
  4617.7  175.42  4696.3  172.82  4781.4  172.29  4909.8  174.67  4953.1  170.27
    4974  169.81    4997  166.37  4999.8  165.87    5003  166.37  5009.2  168.67
  5038.1  170.51  5087.9  169.36  5286.8  171.92    5587  170.38  5907.8  172.05
  6142.2  187.23    6314  202.96  6498.5  211.38  6647.7  211.66    6802  216.42
#Mann= 5 ,-1 , 0
  3891.5      .1       0  4171.7     .05       0  4293.2      .1       0
    4997     .07       0    5003      .1       0
Bank Sta=4974,5038.1
XS Rating Curve= 0 ,0
Exp/Cntr=0.3,0.1

Type RM Length L Ch R = 1 ,34917   ,644,644,644
BEGIN DESCRIPTION:
SALT BRANCH 45.0
END DESCRIPTION:
XS GIS Cut Line= 3
      2235327.42     13322271.76      2235429.06      13321114.2
      2234571.74     13319856.41
#Sta/Elev= 30
  3640.3  184.26  3718.8  182.58  3779.3  180.57  3986.5  175.41  4127.1  175.86
  4155.2  177.33  4257.6   172.6  4307.8  173.69  4327.8  172.01  4418.2   171.9
  4502.3  174.25  4518.6  172.65  4727.1  177.96  4887.2  178.09    4932     175
  4944.3  171.85  4967.9  168.69    4997  164.23  4999.8  163.73    5003  164.23
  5016.9  168.99  5111.6  167.23  5174.5  168.76  5464.6  169.43  5608.2  174.97
  5844.6  180.56  6131.9  197.59  6263.4  203.07  6269.5  204.42  6324.5  205.76
#Mann= 5 ,-1 , 0
  3640.3      .1       0  3718.8     .05       0  3779.3      .1       0
    4997     .07       0    5003      .1       0
Bank Sta=4967.9,5016.9
XS Rating Curve= 0 ,0
Exp/Cntr=0.3,0.1

Type RM Length L Ch R = 1 ,34273   ,800,800,800
BEGIN DESCRIPTION:
Mapping XS ea9b0a17
END DESCRIPTION:
XS GIS Cut Line= 4
      2235570.23     13322164.49      2235621.05     13321035.14
      2235818.69     13320193.77      2235327.43     13319493.58
#Sta/Elev= 30
  3351.5  189.69  3356.1  189.36  3609.4  178.86  3669.5  177.57  3739.5  173.89
  3879.7  171.63  3889.7  170.73  4280.1  172.85  4430.2  171.14  4500.8  171.65
  4603.5  168.21  4644.6  168.02  4662.1  166.77  4675.4  168.15  4752.1  168.92
  4879.3  167.68  4926.8  168.19  4952.8  166.49  4969.2  166.99  4983.6  166.76
    4997  164.04  4999.8  163.54    5003  164.04  5011.7  168.48  5065.7   168.2
  5352.6  171.25  5668.1     171  5760.5  174.02  5989.9  183.94  6201.6  194.72
#Mann= 4 ,-1 , 0
  3351.5     .05       0  3356.1      .1       0    4997     .07       0
    5003      .1       0
Bank Sta=4969.2,5011.7
XS Rating Curve= 0 ,0
Exp/Cntr=0.3,0.1

Type RM Length L Ch R = 1 ,33473   ,522,522,522
BEGIN DESCRIPTION:
SALT BRANCH 44.0
END DESCRIPTION:
XS GIS Cut Line= 3
      2235773.52     13322243.51      2235813.04     13321667.58
      2236552.58     13320521.57
#Sta/Elev= 30
  3849.3  204.02  3987.5  197.55  4006.3  195.09  4016.3  196.21  4145.2  191.33
  4196.8  189.27  4256.9  183.17  4322.6   179.2  4422.1  176.75  4528.6   170.5
  4617.9  167.13  4807.8  164.65  4974.1  165.52    4997   162.6  4999.8   162.1
    5003   162.6  5010.4  162.83  5016.4  165.21  5161.5  169.28  5197.8  171.85
  5203.8  173.76  5234.1  175.31  5240.1  174.19  5255.3  176.42  5261.2  174.62
  5333.8  177.75    5479  188.61  5624.2  196.94  5711.9  205.51  5790.5  220.56
#Mann= 6 ,-1 , 0
  3849.3     .05       0  4145.2      .1       0  4322.6     .05       0
  4528.6      .1       0    4997     .07       0    5003      .1       0
Bank Sta=4974.1,5016.4
XS Rating Curve= 0 ,0
Exp/Cntr=0.3,0.1

Type RM Length L Ch R = 1 ,32951   ,438,438,438
BEGIN DESCRIPTION:
SALT BRANCH 43.0
END DESCRIPTION:
XS GIS Cut Line= 3
      2236037.74     13322046.82      2236237.72     13321696.85
      2236637.72     13320896.85
#Sta/Elev= 30
  4589.1  201.31    4595  201.16  4640.2  198.47  4699.2  191.83    4705   190.3
    4764  185.38  4785.6  180.75  4814.9  178.08  4860.4  174.33  4876.3  171.68
  4911.5  170.27  4978.5  164.76  4984.2  163.81  4989.3  161.24    4995  161.24
    4997  159.65  4999.8  159.15    5003  159.65  5006.1  162.09  5022.9  163.91
  5067.6  165.21  5238.1  164.68  5475.7  169.66  5537.2  172.64  5685.3  176.62
  5693.7  178.19  5699.3  177.57  5716.1  179.41  5730.1  179.45  5886.6  189.97
#Mann= 5 ,-1 , 0
  4589.1      .1       0    4595     .05       0  4814.9      .1       0
    4997     .07       0    5003      .1       0
Bank Sta=4978.5,5022.9
XS Rating Curve= 0 ,0
Exp/Cntr=0.3,0.1

Type RM Length L Ch R = 1 ,32513   ,439,439,439
BEGIN DESCRIPTION:
SALT BRANCH 42.0
END DESCRIPTION:
XS GIS Cut Line= 2
      2236343.82      13322367.8      2237196.48     13320854.48
#Sta/Elev= 30
  4568.7  198.81  4602.7  198.34  4630.2  196.37  4651.9   192.7  4705.4  189.63
  4732.8  185.84  4764.7  185.74  4786.3  181.89    4808  176.55  4906.4  169.11
  4969.8  163.22    4997  160.49  4999.8  159.99    5003  160.49    5006  161.57
  5018.9  162.09  5063.3  162.76  5109.3  163.91  5180.7  163.17  5299.2   165.9
  5423.5  165.95  5585.3  167.89  5709.6  172.19  5833.8  177.54  6033.2  189.09
  6054.9  191.67  6107.8  194.68  6119.9  196.44  6195.1  200.79  6305.7   210.6
#Mann= 5 ,-1 , 0
  4568.7      .1       0  4602.7     .05       0  4906.4      .1       0
    4997     .07       0    5003      .1       0
Bank Sta=4969.8,5063.3
XS Rating Curve= 0 ,0
Exp/Cntr=0.3,0.1

Type RM Length L Ch R = 1 ,32074   ,648,648,648
BEGIN DESCRIPTION:
SALT BRANCH 41.0
END DESCRIPTION:
XS GIS Cut Line= 3
      2236411.56     13322898.61      2236767.34     13322576.71
      2237354.58     13321091.69
#Sta/Elev= 30
  4199.1  195.79  4225.8   196.1  4233.3  194.51  4254.2  194.55  4325.2  189.82
  4360.3  190.05  4452.3  186.02  4622.6  176.02  4665.2  174.79  4675.8  172.95
  4943.4  163.83  4969.9  162.48  4988.9  160.89    4997  158.39  4999.8  157.89
    5003  158.39  5018.7  161.99  5194.9   160.7  5210.6  161.01  5227.2  165.16
  5240.3  165.37  5402.6  165.16  5486.4  163.56  5613.5  166.07  5859.5  176.06
  5943.3  181.48  6021.8  184.39  6227.2  196.32  6273.2  199.56  6275.8  200.92
#Mann= 4 ,-1 , 0
  4199.1     .05       0  4943.4      .1       0    4997     .07       0
    5003      .1       0
Bank Sta=4969.9,5018.7
XS Rating Curve= 0 ,0
Exp/Cntr=0.3,0.1
