--- UNT001 IN SPCR.prj (project) ---

Proj Title=UNT001 IN SPCR Base Level Engineering
Current Plan=p01
Default Exp/Contr=0.3,0.1
English Units
Geom File=g01
Flow File=f01
Plan File=p01
Y Axis Title=Elevation
X Axis Title(PF)=Main Channel Distance
X Axis Title(XS)=Station
BEGIN DESCRIPTION:
UNT001 IN SPCR
END DESCRIPTION:
DSS Export Rating Curves= 0
DSS Export Rating Curve Sorted= 0
DSS Export Volume Flow Curves= 0
DXF OffsetX= 0
DXF OffsetY= 0
DXF ScaleX= 1
DXF ScaleY= 10

--- UNT001 IN SPCR.p01 (plan) ---

Plan Title=Multiple Run
Short Identifier=Multiple
Geom File=g01
Flow File=f01
Subcritical Flow
K Sum by GR= 0
Std Step Tol= 0.01
Critical Tol= 0.01
Num of Std Step Trials= 20
Max Error Tol= 0.3
Flow Tol Ratio= 0.001
Split Flow NTrial= 30
Split Flow Tol= 0.02
Split Flow Ratio= 0.02
Log Output Level= 0
Friction Slope Method= 1
Unsteady Friction Slope Method= 2
Unsteady Bridges Friction Slope Method= 1
Parabolic Critical Depth
Global Vel Dist=  1 , 1 , 1
Global Log Level= 0
CheckData=True
Encroach Param= -1, 0, 0, 0
BEGIN DESCRIPTION:
Multiple Run
END DESCRIPTION:

--- UNT001 IN SPCR.f01 (steady flow) ---

Flow Title=Multiple
Program Version=4.10
Number of Profiles= 7
Profile Names=10-year,25-year,50-year,1pct_min,100-year,1pct_plu,500-year
River Rch & RM=UNT001 IN SPCR,Reach-1         ,29181
     326     467     587     543     735     993    1170
River Rch & RM=UNT001 IN SPCR,Reach-1         ,24145
     460     668     850     794    1074    1452    1743
River Rch & RM=UNT001 IN SPCR,Reach-1         ,23567
     460     668     850     794    1074    1452    1743
River Rch & RM=UNT001 IN SPCR,Reach-1         ,21979
     543     795    1015     952    1287    1741    2103
River Rch & RM=UNT001 IN SPCR,Reach-1         ,19189
     567     828    1055     987    1335    1805    2171
River Rch & RM=UNT001 IN SPCR,Reach-1         ,14064
     778    1150    1478    1393    1883    2547    3109
River Rch & RM=UNT001 IN SPCR,Reach-1         ,13204
     778    1150    1478    1393    1883    2547    3109
River Rch & RM=UNT001 IN SPCR,Reach-1         ,11065
    1024    1528    1974    1870    2529    3420    4218
River Rch & RM=UNT001 IN SPCR,Reach-1         ,10644
    1024    1528    1974    1870    2529    3420    4218
River Rch & RM=UNT001 IN SPCR,Reach-1         ,5834
    1037    1542    1990    1881    2544    3441    4226
Boundary for River Rch & Prof#=UNT001 IN SPCR,Reach-1         , 1
Up Type= 0
Dn Type= 3
Dn Slope=0.005
Boundary for River Rch & Prof#=UNT001 IN SPCR,Reach-1         , 2
Up Type= 0
Dn Type= 3
Dn Slope=0.005
Boundary for River Rch & Prof#=UNT001 IN SPCR,Reach-1         , 3
Up Type= 0
Dn Type= 3
Dn Slope=0.005
Boundary for River Rch & Prof#=UNT001 IN SPCR,Reach-1         , 4
Up Type= 0
Dn Type= 3
Dn Slope=0.005
Boundary for River Rch & Prof#=UNT001 IN SPCR,Reach-1         , 5
Up Type= 0
Dn Type= 3
Dn Slope=0.005
Boundary for River Rch & Prof#=UNT001 IN SPCR,Reach-1         , 6
Up Type= 0
Dn Type= 3
Dn Slope=0.005
Boundary for River Rch & Prof#=UNT001 IN SPCR,Reach-1         , 7
Up Type= 0
Dn Type= 3
Dn Slope=0.005
DSS Import GetInterval= 0
DSS Import GetPeak= 0
DSS Import FillOption= 0

--- UNT001 IN SPCR.g01 (geometry) ---

Geom Title=Existing Conditions
Program Version=4.10

River Reach=UNT001 IN SPCR  ,Reach-1
Reach XY= 30
      2190222.29     13257739.59        2191119.     13258253.96
      2191433.67     13258216.04      2191957.42     13258907.21
      2192168.66     13259369.77      2191911.41     13259946.26
      2192334.78     13260688.07      2192488.96      13262035.2
      2193485.74     13262664.35      2193675.39     13263583.23
      2194929.49     13264520.76      2195625.73     13265482.68
      2195693.28     13266207.68      2196400.29     13266102.18
      2196797.72     13267066.85      2197346.76     13267256.63
      2198396.89     13266544.38      2199023.45     13266485.02
      2199702.97     13267254.11      2199984.79     13268578.81
      2201648.19     13268915.72      2203566.73     13269009.25
      2204395.52     13269801.88      2204911.39     13271020.18
      2205452.41     13270917.31       2205834.2      13271124.4
      2206355.23     13271677.88      2206746.18     13272530.92
      2207378.26     13272866.05      2208202.05      13272788.2

Type RM Length L Ch R = 1 ,29181   ,475,475,475
BEGIN DESCRIPTION:
UNT001 IN SPCR 55.0
END DESCRIPTION:
XS GIS Cut Line= 3
      2190337.74     13258346.81      2190537.72     13257946.85
      2190687.72     13257146.86
#Sta/Elev= 30
  4543.7  397.71  4619.1  395.49  4633.1  394.26  4730.9  390.32  4795.2  388.44
  4901.4  384.64  4923.8  384.62  4954.5  382.71    4998  381.76  5000.8  381.26
    5004  381.76  5041.7  383.15  5092.6  383.09  5255.4   389.2  5290.2  389.49
  5306.3  390.89  5336.8  391.59  5342.7  392.83  5387.7  394.87    5408  394.52
  5433.3  396.25  5558.1  402.85  5570.8  402.78  5652.2  406.19  5692.9  409.37
    5726  410.11  5773.4  414.01  5778.5   413.2  5795.3  414.94  5804.8  415.29
#Mann= 6 ,-1 , 0
  4543.7     .05       0  4795.2      .1       0    4998     .07       0
    5004      .1       0  5433.3     .05       0  5795.3      .1       0
Bank Sta=4954.5,5041.7
XS Rating Curve= 0 ,0
Exp/Cntr=0.3,0.1

Type RM Length L Ch R = 1 ,28706   ,407,407,407
BEGIN DESCRIPTION:
UNT001 IN SPCR 54.0
END DESCRIPTION:
XS GIS Cut Line= 4
      2190698.48      13258539.3      2190915.47     13258278.92
      2191045.68     13257747.24      2191034.83     13257324.02
#Sta/Elev= 30
  4506.8  393.89  4697.1  386.28  4714.1  385.11  4734.9  385.59  4742.8  384.51
  4880.1     380  4963.3  378.51    4992  378.99  5001.9  376.45  5004.6  375.95
  5007.9  376.45  5012.6  378.66  5033.2  379.57  5088.1   378.9  5207.8  381.21
    5213  380.77  5218.5  381.53  5301.3  382.83  5319.4  383.79  5433.5  387.62
  5443.5  388.73  5493.6   390.6  5523.6  392.72  5623.6  396.15  5653.6   396.1
  5663.6  396.66  5673.6  398.53  5693.6   399.5  5703.6  399.13  5816.5  402.78
#Mann= 5 ,-1 , 0
  4506.8     .05       0  4697.1      .1       0  5001.9     .07       0
  5007.9      .1       0  5319.4     .05       0
Bank Sta=4992,5012.6
XS Rating Curve= 0 ,0
Exp/Cntr=0.3,0.1

Type RM Length L Ch R = 1 ,28299   ,487,487,487
BEGIN DESCRIPTION:
UNT001 IN SPCR 53.0
END DESCRIPTION:
XS GIS Cut Line= 3
      2191002.27     13258767.21      2191284.39     13258419.98
       2191306.1     13257584.45
#Sta/Elev= 30
  4325.3  394.08  4358.3  392.64  4378.7  391.32  4436.1  390.03  4442.6  389.11
  4450.5  389.27  4493.3  387.51  4573.8  383.57  4592.7   383.4  4621.5  381.22
    4671   380.1  4677.5  379.34  4699.4  378.64  4806.7  376.72  4895.9  376.53
  4915.9  377.15  4925.9  376.53  5002.9  376.25  5005.6  375.75  5008.9  376.25
  5065.9  377.12  5086.9  377.47  5118.1  377.73    5196  379.45    5226   379.1
    5246  380.31    5256  379.96    5326  380.97  5416.9  383.57  5608.5  388.88
#Mann= 9 ,-1 , 0
  4325.3      .1       0  4358.3     .05       0  4573.8      .1       0
  4806.7     .08       0  5002.9     .07       0  5008.9     .08       0
  5086.9      .1       0  5118.1     .05       0  5416.9      .1       0
Bank Sta=4915.9,5065.9
XS Rating Curve= 0 ,0
Exp/Cntr=0.3,0.1

Type RM Length L Ch R = 1 ,27812   ,465,465,465
BEGIN DESCRIPTION:
UNT001 IN SPCR 52.0
END DESCRIPTION:
XS GIS Cut Line= 3
      2191087.72     13259096.85      2191637.72     13258446.85
      2192037.75     13258296.84
#Sta/Elev= 30
  4166.3  400.65  4237.2  398.76    4258  397.35  4328.6  394.73  4400.9  391.57
  4415.2  391.56  4442.6  389.25  4493.2  387.43  4506.9  385.72  4542.6   385.4
  4553.6  384.47  4677.2  378.75  4727.2  377.72  4755.8  375.93  4883.2  373.73
  4923.1  372.78  4925.8  372.28  4929.1  372.78    4982  373.41    5113   373.3
  5143.3  373.89  5167.3  376.49  5203.8  377.44  5252.7  380.17  5289.2  380.17
  5295.4  381.41  5306.1  381.46  5319.5  382.78  5344.4  383.53    5445  389.37
#Mann= 5 ,-1 , 0
  4166.3      .1       0  4328.6     .05       0  4553.6      .1       0
  4923.1     .07       0  4929.1      .1       0
Bank Sta=4883.2,4982
XS Rating Curve= 0 ,0
Exp/Cntr=0.3,0.1

Type RM Length L Ch R = 1 ,27347   ,423,423,423
BEGIN DESCRIPTION:
UNT001 IN SPCR 51.0
END DESCRIPTION:
XS GIS Cut Line= 3
      2191284.38     13259103.58      2191653.32     13258973.37
       2192293.1     13258474.55
#Sta/Elev= 30
  4380.7  394.94  4387.7  395.22  4413.3  393.86  4444.3     391  4458.5  392.11
  4469.1  391.88  4531.8  389.88  4543.3  388.49  4556.6  388.14  4598.9  385.31
  4617.5  385.19  4685.9  381.55  4702.4  381.38    4712   380.1  4748.3  378.06
    4766  378.03  4942.9  371.09  4997.8  369.89  5000.5  369.39  5003.8  369.89
  5007.1  370.43  5050.5  370.32  5056.9  371.01    5150  373.62  5249.5  379.65
  5413.3  387.56  5456.7  390.79  5506.5  393.21    5513  394.22  5583.2  397.09
#Mann= 5 ,-1 , 0
  4380.7      .1       0  4556.6     .05       0  4685.9      .1       0
  4997.8     .07       0  5003.8      .1       0
Bank Sta=4942.9,5056.9
XS Rating Curve= 0 ,0
Exp/Cntr=0.3,0.1

Type RM Length L Ch R = 1 ,26924   ,518,518,518
BEGIN DESCRIPTION:
UNT001 IN SPCR 50.0
END DESCRIPTION:
XS GIS Cut Line= 4
      2191414.59     13259212.08      2191837.78     13259212.08
      2192250.11     13259071.02       2192390.9     13258681.14
#Sta/Elev= 30
  4326.2  389.22  4379.3  387.76  4389.3   386.5  4419.3  384.81  4449.3  385.44
  4459.3  384.29  4479.3  383.82  4489.3  384.39  4499.3  383.11  4519.3  382.94
  4539.3  381.27  4609.3   379.1  4669.3   375.6  4749.4  374.04  4770.5  372.71
  4791.6  372.52  4886.7  368.99  4960.7   368.6  4992.2  367.68  4997.5  368.35
    5000  367.16  5002.7  366.66    5006  367.16  5013.6  368.17  5034.7  368.87
  5243.5  376.36  5280.6  378.65  5317.2  379.82  5367.3  382.65  5599.7  392.82
#Mann= 4 ,-1 , 0
  4326.2      .1       0    5000     .07       0    5006      .1       0
  5243.5     .05       0
Bank Sta=4960.7,5034.7
XS Rating Curve= 0 ,0
Exp/Cntr=0.3,0.1

Type RM Length L Ch R = 1 ,26406   ,444,444,444
BEGIN DESCRIPTION:
UNT001 IN SPCR 49.0
END DESCRIPTION:
XS GIS Cut Line= 4
      2191382.02     13259374.82      2191653.32      13259559.3
      2192358.61     13259526.75       2192879.4     13259418.25
#Sta/Elev= 30
  4288.1  387.08  4415.9  382.49  4459.5     380  4524.8  377.86  4531.3  376.91
  4552.3  376.69  4650.6  372.72  4770.7  369.57  4781.7  370.19  4810.8   369.3
  4870.9  369.32  4940.9  367.43    4978  366.08  4980.7  365.58    4984  366.08
  5111.1  367.54  5121.1  367.98  5141.1   366.8  5171.2  367.39  5208.9  366.91
  5221.2  367.54  5362.2  368.31  5446.6  370.34  5491.6  372.26  5591.3  375.05
  5627.8  377.03  5641.7  376.85  5678.8  378.08  5818.5  383.95  5854.2   385.1
#Mann= 5 ,-1 , 0
  4288.1      .1       0    4978     .07       0    4984      .1       0
  5591.3     .05       0  5818.5      .1       0
Bank Sta=4940.9,5111.1
XS Rating Curve= 0 ,0
Exp/Cntr=0.3,0.1

Type RM Length L Ch R = 1 ,25962   ,560,560,560
BEGIN DESCRIPTION:
UNT001 IN SPCR 48.0
END DESCRIPTION:
XS GIS Cut Line= 4
      2191284.36     13259895.67      2191664.17     13259982.48
      2192282.66     13259852.27      2192878.54     13259581.42
#Sta/Elev= 30
  4354.6  391.16  4399.1  389.73  4431.1  387.34  4474.1  386.52  4602.9  379.06
  4614.5  379.33  4665.8  375.85  4717.1  374.37  4744.2  372.11  4813.8  369.03
  4823.3  368.41    4850  368.37  4946.6  364.24  4962.4  363.94    4986  362.54
  4988.7  362.04    4992  362.54  4994.1  363.51  5023.8  363.92  5289.5  364.34
  5332.6  362.69  5371.2  364.92  5422.9  364.59  5513.6  366.17  5634.5   369.7
  5669.1  371.72    5731  373.72  5912.8  381.59  5934.8  381.56  6030.8  385.87
#Mann= 9 ,-1 , 0
  4354.6      .1       0  4813.8     .08       0  4823.3     .05       0
  4946.6      .1       0    4986     .07       0    4992      .1       0
  5669.1     .05       0    5731      .1       0  5912.8     .05       0
Bank Sta=4962.4,5023.8
XS Rating Curve= 0 ,0
Exp/Cntr=0.3,0.1

Type RM Length L Ch R = 1 ,25402   ,463,463,463
BEGIN DESCRIPTION:
UNT001 IN SPCR 47.0
END DESCRIPTION:
XS GIS Cut Line= 4
      2191392.91     13260232.05      2191685.87     13260373.11
      2192434.57      13260329.7      2193020.47      13259787.2
#Sta/Elev= 30
  4195.7  387.15  4256.5  384.45  4263.2  383.21  4285.9  382.46  4291.4  383.29
  4400.5  376.78  4411.9  375.78  4427.2  376.24  4434.1     375  4511.8  371.69
  4524.3  372.07  4540.1  370.39    4673  364.41  4783.1  360.74  4843.2   359.4
  4893.3  360.66  4958.5  360.23  4983.5  360.43  4990.5  359.33  4993.2  358.83
  4996.5  359.33  5013.5  360.95    5057  360.87  5236.3  362.32  5515.7  368.68
  5621.8  368.75  5837.9  377.14  5910.9  380.46  5989.8  383.95  6069.3  387.55
#Mann= 9 ,-1 , 0
  4195.7     .05       0  4400.5      .1       0  4958.5     .05       0
  4990.5     .04       0  4996.5     .05       0    5057      .1       0
  5837.9     .05       0  5910.9      .1       0  5989.8     .05       0
Bank Sta=4983.5,5013.5
XS Rating Curve= 0 ,0
Exp/Cntr=0.3,0.1

Type RM Length L Ch R = 1 ,24939   ,353,353,353
BEGIN DESCRIPTION:
UNT001 IN SPCR 46.0
END DESCRIPTION:
XS GIS Cut Line= 3
      2191458.04     13260666.08      2191978.84     13260774.58
      2192933.25     13260709.51
#Sta/Elev= 30
  4097.5  384.06  4209.5  378.08  4240.2  377.75  4250.4  376.19    4281  376.06
  4316.9  373.91  4352.5  371.53  4369.4  371.01  4374.5  371.71  4419.5  369.63
  4424.6   370.3  4505.8  366.29  4519.6  366.73  4614.6  362.62  4738.6  359.07
  4989.2  357.34  4996.2  356.61    4999  356.11  5002.2  356.61  5029.3   357.6
  5155.6   363.7  5209.7  365.72  5254.2  368.62  5289.9  369.99    5330  370.02
    5340  370.75    5350  373.23  5404.9  374.73  5540.5  382.07  5586.1  382.96
#Mann= 6 ,-1 , 0
  4097.5     .05       0  4316.9      .1       0  4996.2     .07       0
  5002.2      .1       0  5155.6     .08       0  5254.2     .05       0
Bank Sta=4989.2,5029.3
XS Rating Curve= 0 ,0
Exp/Cntr=0.3,0.1

Type RM Length L Ch R = 1 ,24586   ,441,441,441
BEGIN DESCRIPTION:
UNT001 IN SPCR 45.0
END DESCRIPTION:
XS GIS Cut Line= 3
      2191587.68     13260946.85      2192387.72     13261096.85
      2192787.73     13260946.85
#Sta/Elev= 30
  4193.7  379.69    4220  377.96  4330.2  374.59  4417.6  370.37  4440.5  369.97
  4468.4  367.62  4509.1  365.82  4691.6  359.49  4743.2  357.38  4981.4  355.67
  4987.3   354.2  4994.5   353.8  4997.3   353.3  5000.5   353.8  5010.4  354.34
  5017.5  355.62  5061.1  356.06  5093.1  357.95  5157.2  360.22  5218.6  363.88
  5242.6  365.64  5254.2  367.33  5273.8  367.38  5333.5  370.55  5349.4  370.95
  5370.8  372.74  5389.5  373.32  5394.8  374.26  5413.5  374.63  5434.9  376.19
#Mann= 5 ,-1 , 0
  4193.7     .05       0  4691.6      .1       0  4994.5     .07       0
  5000.5      .1       0  5333.5     .08       0
Bank Sta=4981.4,5017.5
XS Rating Curve= 0 ,0
Exp/Cntr=0.3,0.1

Type RM Length L Ch R = 1 ,24145   ,578,578,578
BEGIN DESCRIPTION:
UNT001 IN SPCR 44.0
END DESCRIPTION:
XS GIS Cut Line= 2
      2191838.11     13261951.86      2193046.45     13261113.31
#Sta/Elev= 30
  4140.4  364.68  4322.5  359.38  4351.9  359.39  4417.4  356.55  4585.6  354.18
  4611.3  353.12  4632.2  354.27    4668  354.32  4754.5  353.83  4784.2  352.86
  4805.1  353.81  4918.9  354.36  4955.5  353.76    4978  354.52    4992  353.67
    4996  351.88  4998.7  351.38    5002  351.88  5013.8  353.98  5019.9  354.08
  5028.5  355.25  5055.7  355.11  5127.3  357.44  5243.5  362.82    5336  365.87
  5344.8  366.91  5430.2  370.19  5496.5  373.91  5567.6  377.77  5611.2  379.26
#Mann= 6 ,-1 , 0
  4140.4     .05       0  4585.6      .1       0    4996     .07       0
    5002      .1       0  5496.5     .08       0  5567.6      .1       0
#XS Ineff= 1 ,-1
 4562.05 4662.74  354.31
Permanent Ineff=
       F
Bank Sta=4978,5019.9
XS Rating Curve= 0 ,0
Exp/Cntr=0.3,0.1

Type RM Length L Ch R = 1 ,23567   ,387,387,387
BEGIN DESCRIPTION:
UNT001 IN SPCR 43.0
END DESCRIPTION:
XS GIS Cut Line= 2
      2192114.14     13262311.24      2193202.69     13261342.48
#Sta/Elev= 30
  4522.3  367.09  4584.4  364.81  4606.2  363.24  4641.3   362.5  4669.7  360.88
  4676.4  361.26  4690.6  359.96  4704.8  359.89  4832.8  354.19  4953.2  351.83
    4963  351.51  4992.6   350.4  4995.4   349.9  4998.6   350.4  5030.9  351.56
  5073.6  351.29  5151.4  352.61  5222.4  352.25  5342.8  354.39    5378  356.64
  5398.9  356.51  5526.8  362.84  5533.5  362.47  5682.3  368.39  5689.8  369.68
  5739.2  371.22  5824.5  375.31  5859.6  377.93    5887  378.69  5979.5  382.83
#Mann= 5 ,-1 , 0
  4522.3     .05       0    4963      .1       0  4992.6     .07       0
  4998.6      .1       0    5887     .08       0
Bank Sta=4953.2,5030.9
XS Rating Curve= 0 ,0
Exp/Cntr=0.3,0.1

Type RM Length L Ch R = 1 ,23180   ,291,291,291
BEGIN DESCRIPTION:
UNT001 IN SPCR 42.0
END DESCRIPTION:
XS GIS Cut Line= 3
      2192387.74     13262646.83      2192737.72     13262246.85
      2193437.72     13261446.85
#Sta/Elev= 30
  4500.3  373.69  4550.1   370.1  4585.2   369.7  4599.5  368.43  4606.6  365.95
  4620.3  364.34  4627.9  365.23  4663.7  364.51  4854.8     355  4930.7  352.14
  4961.1   350.4  4989.5     349  4993.2  348.02  4995.9  347.52  4999.2  348.02
  5024.7  349.92  5151.8  349.87  5435.6  356.31  5627.4  365.23  5683.4  367.12
  5803.9  373.52  5846.6  374.96  5854.2  376.35  5860.8  375.82  5881.6  376.66
  5946.3  381.05  6030.7  385.11    6045  384.86  6073.4  387.36  6094.8  387.62
#Mann= 7 ,-1 , 0
  4500.3     .08       0  4663.7     .05       0  4930.7      .1       0
  4993.2     .07       0  4999.2      .1       0  5881.6     .08       0
  6030.7      .1       0
Bank Sta=4961.1,5024.7
XS Rating Curve= 0 ,0
Exp/Cntr=0.3,0.1

Type RM Length L Ch R = 1 ,22889   ,319,319,319
BEGIN DESCRIPTION:
Mapping XS a9a7feac
END DESCRIPTION:
XS GIS Cut Line= 3
      2192486.83     13262749.05      2192905.96     13262477.49
      2193571.84     13261640.72
#Sta/Elev= 30
  4396.3  374.91  4572.6  366.46  4578.5   365.4  4593.7  365.73  4608.9  364.87
  4614.8  362.82  4635.9  360.69  4649.1  360.81  4681.4  359.65  4702.5  360.57
  4913.5  350.55  4960.8  348.99    5001  347.85  5003.8  347.35    5007  347.85
  5018.5  348.67    5318   351.7  5353.2  354.09  5409.3  354.71  5587.1  361.79
    5688  367.28  5694.4  366.59  5729.6  369.12    5744  368.14  5758.5  368.65
  5787.3  372.41  5820.1  373.47  5917.9  377.04  5929.9  377.96  5965.1  377.32
#Mann= 7 ,-1 , 0
  4396.3     .08       0  4649.1     .05       0  4913.5      .1       0
    5001     .07       0    5007      .1       0  5820.1     .08       0
  5917.9      .1       0
Bank Sta=4960.8,5018.5
XS Rating Curve= 0 ,0
Exp/Cntr=0.3,0.1

Type RM Length L Ch R = 1 ,22570   ,241,241,241
BEGIN DESCRIPTION:
Mapping XS 5dfc348b
END DESCRIPTION:
XS GIS Cut Line= 3
      2192510.55     13262803.65       2192998.8     13262564.95
       2194104.1     13262326.55
#Sta/Elev= 30
  4197.5   375.6  4461.5  364.11  4483.8  361.87    4516  361.78  4521.5  359.66
  4528.3   358.7  4570.5  357.23  4628.5  357.15  4639.7  355.93    4743  352.88
  4760.5  351.45  4799.6  351.27  4804.7   350.3  4862.6  348.46  4918.9  347.76
  4947.5  347.92  4961.9  346.45  4964.7  345.95  4967.9  346.45  5085.1  348.28
  5128.6   348.5  5261.6  353.12  5599.2  372.08  5650.3  374.01  5656.1  375.59
  5700.3  376.69  5705.4  377.89  5793.6  381.03    5814  382.66  5871.7  383.37
#Mann= 5 ,-1 , 0
  4197.5     .08       0  4570.5     .05       0  4918.9      .1       0
  4961.9     .07       0  4967.9      .1       0
Bank Sta=4947.5,5085.1
XS Rating Curve= 0 ,0
Exp/Cntr=0.3,0.1

Type RM Length L Ch R = 1 ,22329   ,350,350,350
BEGIN DESCRIPTION:
Mapping XS 47fca5ed
END DESCRIPTION:
XS GIS Cut Line= 3
      2192618.99     13262825.38      2193183.27     13262608.35
      2194093.72     13262727.57
#Sta/Elev= 30
    4125  372.18  4175.7   369.9  4271.2  365.42  4276.5  365.97  4284.3  364.76
  4348.6  361.82  4402.2   360.4  4440.5   357.7  4465.1  357.86  4477.2  355.63
  4500.5   354.4  4563.5   353.6  4585.1  353.81  4705.1  349.77  4831.7  347.24
  4925.7  346.92  4973.1  345.75  4975.9  345.25  4979.1  345.75  5063.2  346.85
  5068.3  346.08  5117.3  347.42  5177.8  350.85  5228.2  351.87  5294.7  355.94
  5299.8  355.14    5430  361.49  5452.4  361.34  5526.2   365.9  5647.8  369.48
#Mann= 6 ,-1 , 0
    4125     .05       0  4175.7     .08       0  4563.5     .05       0
  4705.1      .1       0  4973.1     .07       0  4979.1      .1       0
Bank Sta=4925.7,5063.2
XS Rating Curve= 0 ,0
Exp/Cntr=0.3,0.1

Type RM Length L Ch R = 1 ,21979   ,127,127,127
BEGIN DESCRIPTION:
Mapping XS 6edfa7e2
END DESCRIPTION:
XS GIS Cut Line= 3
      2192619.07     13262890.46      2193139.86     13262847.06
      2194409.37     13263096.62
#Sta/Elev= 30
  3998.4  371.97  4157.6  367.28  4167.6  365.92    4268  361.67  4330.2  360.17
  4458.5  354.99  4620.7  350.33  4630.9  349.07  4722.6   349.6  4773.6   347.1
    4807  347.26  4906.5  346.63  4926.5  346.79  4984.6  345.88  4987.4  345.38
  4990.6  345.88    5059  347.03  5109.9  347.19  5130.3  348.32  5150.7  351.09
  5181.3   350.2  5252.6   354.1  5304.4  355.06  5391.4  356.95    5538  358.72
  5686.1  363.18  5711.2  362.85  5737.5  365.02  5742.6  364.18  5814.8  366.17
#Mann= 8 ,-1 , 0
  3998.4     .05       0  4330.2     .08       0    4807      .1       0
  4906.5     .08       0  4984.6     .07       0  4990.6     .08       0
  5304.4      .1       0  5391.4     .08       0
Bank Sta=4926.5,5059
XS Rating Curve= 0 ,0
Exp/Cntr=0.3,0.1

Type RM Length L Ch R = 1 ,21852   ,240,240,240
BEGIN DESCRIPTION:
Mapping XS df2068ec
END DESCRIPTION:
XS GIS Cut Line= 4
      2192640.77     13262966.43      2193302.62     13263042.38
      2193801.75     13263074.93      2194279.14     13263140.03
#Sta/Elev= 30
  4002.3   369.7  4059.6  367.55    4110  367.14  4190.5  364.04  4220.5   364.1
  4230.7  362.67  4319.7  360.34  4398.1  358.05  4603.2   352.2  4633.4  350.24
  4743.8  348.53  4792.2  346.49  4833.9  345.27    4864  346.05  4984.3  345.43
  5011.3  344.74  5014.1  344.24  5017.3  344.74  5034.4  345.95  5084.5  345.24
  5114.5  347.38    5215  350.99  5336.2   353.2  5346.3  354.37    5427  354.53
    5437   355.5  5467.4  355.89  5497.7  357.42  5546.2  358.08  5650.5  362.12
#Mann= 7 ,-1 , 0
  4002.3     .05       0  4319.7      .1       0  4398.1     .05       0
  4792.2      .1       0  5011.3     .07       0  5017.3      .1       0
  5546.2     .08       0
Bank Sta=4984.3,5034.4
XS Rating Curve= 0 ,0
Exp/Cntr=0.3,0.1

Type RM Length L Ch R = 1 ,21612   ,315,315,315
BEGIN DESCRIPTION:
Mapping XS a23436fc
END DESCRIPTION:
XS GIS Cut Line= 3
      2192597.36     13263508.95      2193226.67      13263367.9
      2194244.67     13263205.45
#Sta/Elev= 30
  3911.8  369.02  3973.7  366.56  3983.9  366.98  3994.6  365.58  4095.5  361.87
    4265  356.23  4270.9  355.39  4332.3  354.22  4351.7  352.91  4356.8  353.77
  4443.6  352.14  4448.7  352.93    4492  351.63  4588.2  352.12  4618.5  350.72
  4661.3  351.24  4710.1  350.21  4750.2  350.16  4796.2  347.84  4922.3  344.43
  4993.2  344.05  5000.4  343.32  5003.1  342.82  5006.4  343.32  5023.6  344.49
  5033.7  343.85  5354.6  351.49  5478.9  355.23  5529.9  358.13  5587.6  360.07
#Mann= 6 ,-1 , 0
  3911.8     .05       0  4095.5      .1       0  4710.1     .05       0
  4796.2      .1       0  5000.4     .07       0  5006.4      .1       0
Bank Sta=4993.2,5023.6
XS Rating Curve= 0 ,0
Exp/Cntr=0.3,0.1

Type RM Length L Ch R = 1 ,21297   ,511,511,511
BEGIN DESCRIPTION:
UNT001 IN SPCR 38.0
END DESCRIPTION:
XS GIS Cut Line= 3
      2193098.02     13263947.63      2193429.48     13263751.21
      2194233.63     13263249.89
#Sta/Elev= 30
  4314.8  364.96  4354.4   363.7  4366.1  363.03  4381.7  363.24  4387.5  362.44
  4395.8  362.79  4440.2  360.42  4498.6  359.12  4504.5  358.34  4584.4  354.86
  4615.6  354.57  4621.4  353.63  4651.5  352.69  4658.5  353.11  4679.9  351.58
  4722.6  350.38    4738  348.98  4805.3  347.06  4957.3  343.11  4984.6   344.2
  4996.9  343.05  4999.7  342.55  5002.9  343.05  5021.1  343.75  5036.5  343.25
  5100.2  344.28  5145.8  344.18    5289  346.32  5493.1  353.04  5647.7  359.38
#Mann= 5 ,-1 , 0
  4314.8      .1       0  4354.4     .05       0  4805.3      .1       0
  4996.9     .07       0  5002.9      .1       0
Bank Sta=4984.6,5021.1
XS Rating Curve= 0 ,0
Exp/Cntr=0.3,0.1

Type RM Length L Ch R = 1 ,20786   ,96,96,96
BEGIN DESCRIPTION:
Mapping XS 5b483869
END DESCRIPTION:
XS GIS Cut Line= 3
      2193480.45     13264247.01       2194006.5      13263991.8
      2194209.63     13263476.15
#Sta/Elev= 30
  4340.7  372.27  4353.4  372.68  4359.9  371.28  4398.6  369.46  4421.1  367.19
  4466.3  364.71  4471.8  365.18  4526.6  361.23  4556.6  361.09  4584.7  357.67
  4601.7  358.44  4652.4  354.55  4697.5  353.27  4714.5  351.51  4753.1  350.01
  4915.6  340.85  4930.7  340.86  4939.2  339.37  4962.9  338.84  5013.7  337.15
  5016.4  336.65  5019.7  337.15  5038.2  339.09  5052.9  340.45  5059.7   343.7
  5070.4  343.69  5082.7  341.26  5107.1  343.09  5136.8  342.28  5479.6  354.12
#Mann= 4 ,-1 , 0
  4340.7     .05       0  4753.1      .1       0  5013.7     .07       0
  5019.7      .1       0
Bank Sta=4962.9,5038.2
XS Rating Curve= 0 ,0
Exp/Cntr=0.3,0.1

Type RM Length L Ch R = 1 ,20690   ,70,70,70
BEGIN DESCRIPTION:
Mapping XS 9ccab76c
END DESCRIPTION:
XS GIS Cut Line= 3
      2193615.91     13264293.87      2194063.79     13264069.93
      2194365.86     13263444.95
#Sta/Elev= 30
  4384.5   367.6  4435.3  364.35  4474.4  363.59  4509.5  360.04  4547.1  359.36
  4554.2  357.61  4733.7  348.97  4793.1  347.24  4815.4  344.63  4837.8  344.06
  4854.5  346.14  4860.1  344.61  4867.3  346.92  4882.5  345.92  4884.7  343.84
  4966.4  346.62  4973.3  345.46  5001.5  346.78    5033  343.37  5063.7  345.92
  5077.5  342.69  5088.9  338.47  5091.6  337.97  5094.9  338.47  5108.9  341.87
  5131.5  340.59  5154.1  341.53  5159.7  343.27  5176.7  344.28  5579.4  360.22
#Mann= 4 ,-1 , 0
  4384.5     .05       0  4733.7      .1       0  5088.9     .07       0
  5094.9      .1       0
Bank Sta=4966.4,5001.5
XS Rating Curve= 0 ,0
Exp/Cntr=0.3,0.1

Type RM Length L Ch R = 1 ,20620   ,192,192,192
BEGIN DESCRIPTION:
Mapping XS fb8ab67f
END DESCRIPTION:
XS GIS Cut Line= 4
      2193693.44     13264328.21      2194076.06     13264158.39
      2194209.06     13263943.54      2194438.23     13263495.43
#Sta/Elev= 30
  4405.9  364.69  4424.3  364.32  4442.1  361.82  4465.3  360.19  4592.6  355.02
  4607.5  353.35  4644.6   352.7  4651.3  351.42  4731.9  348.68  4812.9   345.3
  4849.8  344.89  4892.6  342.48  4950.5  342.09  4979.2  342.89  5050.9  342.33
  5060.4  340.95  5063.3  339.15    5066  338.65  5069.3  339.15  5077.2   339.2
  5087.8  341.75  5104.4  341.42    5110  342.42  5253.2   346.8  5309.9  350.39
  5320.6  350.18  5520.8  358.37    5534  359.99  5543.3  359.66  5580.5  361.61
#Mann= 5 ,-1 , 0
  4405.9     .05       0  4731.9      .1       0  5063.3     .07       0
  5069.3      .1       0  5543.3     .05       0
Bank Sta=4979.2,5050.9
XS Rating Curve= 0 ,0
Exp/Cntr=0.3,0.1

Type RM Length L Ch R = 1 ,20428   ,364,364,364
BEGIN DESCRIPTION:
Mapping XS 3680476f
END DESCRIPTION:
XS GIS Cut Line= 3
      2193714.83     13264351.18      2194417.96     13264101.18
      2194735.42     13263601.56
#Sta/Elev= 30
  4376.9  363.16    4571  353.27  4592.2  352.46  4610.9  353.09  4672.6  349.08
  4687.8  349.19  4717.8  347.43  4826.8  344.53  4852.4   342.9  4963.7  340.81
  4998.3  340.14    5001  339.64  5004.3  340.14  5026.8  340.77  5154.3  341.71
  5278.8  344.94  5284.7  344.44    5294  345.36    5306  344.85  5342.3   347.4
  5415.1  349.27  5445.6  352.07    5488  352.67  5545.6  356.22    5582  356.88
  5597.2   358.3  5618.4  357.92  5633.6   359.3  5654.8  359.21  5715.1  362.29
#Mann= 4 ,-1 , 0
  4376.9     .05       0  4717.8      .1       0  4998.3     .07       0
  5004.3      .1       0
Bank Sta=4963.7,5026.8
XS Rating Curve= 0 ,0
Exp/Cntr=0.3,0.1

Type RM Length L Ch R = 1 ,20064   ,436,436,436
BEGIN DESCRIPTION:
UNT001 IN SPCR 35.0
END DESCRIPTION:
XS GIS Cut Line= 3
      2193787.68     13264496.86      2194587.72     13264346.85
      2194987.74     13263946.83
#Sta/Elev= 30
  4168.2  360.51  4178.4  360.49  4219.1  358.01  4239.5  358.47  4247.1  357.69
    4270  357.05  4280.2  355.83  4290.3  355.96  4310.7  354.31    4331  353.44
  4357.3  353.17  4362.4  352.56  4392.1  351.81  4409.9  350.65  4464.7  348.69
    4565  345.46  4572.7  344.75  4646.4  342.72  4758.3  340.85  4890.6  339.89
  4950.8  338.88  4976.6  337.59  4979.4  337.09  4982.6  337.59  5052.9  338.32
  5081.2  338.24  5137.7  339.57    5265  344.38  5448.9  354.35  5547.9  360.97
#Mann= 4 ,-1 , 0
  4168.2     .05       0  4464.7      .1       0  4976.6     .07       0
  4982.6      .1       0
Bank Sta=4950.8,5052.9
XS Rating Curve= 0 ,0
Exp/Cntr=0.3,0.1

Type RM Length L Ch R = 1 ,19628   ,439,439,439
BEGIN DESCRIPTION:
UNT001 IN SPCR 34.0
END DESCRIPTION:
XS GIS Cut Line= 3
      2194537.72     13265196.86      2194937.72     13264546.85
      2195237.71     13264146.87
#Sta/Elev= 30
  4232.3  356.28  4255.4   355.7  4261.3  356.32  4267.5  355.31  4313.4  354.05
    4356  351.73  4377.2  351.55  4508.6  344.58    4590   341.9  4631.5  340.03
  4734.6  337.69  4835.2  337.47  4856.5  336.28  4878.1   337.4    4924  336.99
  4957.3  335.34    4960  334.84  4963.3  335.34  4998.6   335.5  5023.6  336.65
  5145.5  343.79  5152.8  344.93  5173.6  344.96  5217.4  348.29  5338.2  350.97
  5388.2  353.11  5402.8   354.8  5423.6  358.83  5438.2  358.73  5495.5  362.48
#Mann= 4 ,-1 , 0
  4232.3     .05       0    4590      .1       0  4957.3     .07       0
  4963.3      .1       0
Bank Sta=4924,5023.6
XS Rating Curve= 0 ,0
Exp/Cntr=0.3,0.1

Type RM Length L Ch R = 1 ,19189   ,368,368,368
BEGIN DESCRIPTION:
UNT001 IN SPCR 33.0
END DESCRIPTION:
XS GIS Cut Line= 3
       2194604.7     13265396.98      2194908.53     13265201.66
      2195493.62     13264508.21
#Sta/Elev= 30
  4275.7  353.01  4282.8  352.99  4300.4  352.29    4315   352.7  4336.7  351.23
  4350.6  351.47  4357.9  350.55    4373  350.35    4379     351  4386.3   350.1
  4430.5  348.79  4445.7  349.08  4503.2  346.45  4575.8  344.35  4602.9  344.61
  4612.1  343.24  4633.3  342.45  4743.2  340.09  4786.9  338.28  4874.1  335.71
  4972.9  334.43  4980.7  333.67  4987.2  331.12    4992  331.05  4994.7  330.55
    4998  331.05  5009.3  332.14  5015.8   334.3  5299.3  341.24  5544.2  350.74
#Mann= 6 ,-1 , 0
  4275.7     .05       0  4282.8      .1       0  4743.2     .05       0
  4786.9      .1       0    4992     .07       0    4998      .1       0
Bank Sta=4972.9,5015.8
XS Rating Curve= 0 ,0
Exp/Cntr=0.3,0.1

Type RM Length L Ch R = 1 ,18821   ,518,518,518
BEGIN DESCRIPTION:
UNT001 IN SPCR 32.0
END DESCRIPTION:
XS GIS Cut Line= 3
      2194713.21     13265613.99      2195125.54     13265407.83
      2195798.25     13264832.77
#Sta/Elev= 30
  4286.2  349.09  4293.9  347.87  4310.7  348.58  4377.8  345.89  4383.4  346.32
    4398  345.14  4601.4  339.09  4629.3  339.05  4668.4  337.78    4674  338.33
  4745.6  336.37  4912.4  334.96  4955.2  333.73    4995  332.79  4997.8  332.29
    5001  332.79  5039.7  333.47    5054   332.8  5111.1  334.03  5168.2  333.84
  5182.5  334.43    5189  333.99  5281.3  336.41  5373.5  341.54  5387.7  341.74
    5402  342.98  5459.1  344.98  5500.8  347.35  5515.1  347.33  5632.2  353.89
#Mann= 4 ,-1 , 0
  4286.2     .05       0    4398      .1       0    4995     .07       0
    5001      .1       0
Bank Sta=4955.2,5039.7
XS Rating Curve= 0 ,0
Exp/Cntr=0.3,0.1

Type RM Length L Ch R = 1 ,18303   ,465,465,465
BEGIN DESCRIPTION:
UNT001 IN SPCR 31.0
END DESCRIPTION:
XS GIS Cut Line= 3
      2194837.74     13266096.84      2195637.72     13265596.85
      2195837.74     13265446.84
#Sta/Elev= 30
  4047.4  350.07  4097.5  348.87  4200.7   342.9  4236.1  342.51  4248.7  341.48
  4307.4  339.95  4395.8  335.53  4411.4  335.26    4469  333.15    4548  331.87
  4563.3  332.55  4621.1  331.65  4809.8  332.54    4910  330.65  4946.6  330.97
  4983.1  329.83  4987.8  328.25  4993.9  328.25  5001.3  327.32  5004.1  326.82
  5007.3  327.32  5012.6  329.74  5048.1  333.14  5054.3  332.94  5077.2  334.78
  5140.8  337.63  5148.1  338.66  5162.6  339.51  5168.9  339.29  5240.8  343.64
#Mann= 5 ,-1 , 0
  4047.4      .1       0  4248.7     .05       0  4411.4      .1       0
  5001.3     .07       0  5007.3      .1       0
Bank Sta=4983.1,5012.6
XS Rating Curve= 0 ,0
Exp/Cntr=0.3,0.1

Type RM Length L Ch R = 1 ,17838   ,381,381,381
BEGIN DESCRIPTION:
UNT001 IN SPCR 30.0
END DESCRIPTION:
XS GIS Cut Line= 3
      2195337.74     13266796.82      2195687.72     13266046.85
      2196037.71     13265646.87
#Sta/Elev= 30
  4177.1  358.37  4214.1  357.24  4305.5  351.74  4328.4  351.82    4397  347.77
  4408.8  348.24  4516.8  341.49  4682.2  334.81    4773  331.26  4876.2   329.1
  4938.5  329.36  4967.7  330.23  4977.1  328.23  4998.9   325.9  5001.7   325.4
  5004.9   325.9  5011.8  326.05  5018.5  329.92  5032.7  330.44  5103.9  329.42
  5267.1  331.99  5387.7  336.11  5408.6  336.28  5457.9  338.08  5465.5  338.96
  5486.4  338.94  5508.2  340.56  5529.1   340.9  5532.9  342.12  5536.2  342.12
#Mann= 4 ,-1 , 0
  4177.1     .05       0  4682.2      .1       0  4998.9     .07       0
  5004.9      .1       0
Bank Sta=4967.7,5018.5
XS Rating Curve= 0 ,0
Exp/Cntr=0.3,0.1

Type RM Length L Ch R = 1 ,17457   ,544,544,544
BEGIN DESCRIPTION:
UNT001 IN SPCR 29.0
END DESCRIPTION:
XS GIS Cut Line= 3
      2195516.17     13266883.52      2195787.43     13266449.49
      2196264.86     13265624.85
#Sta/Elev= 30
    4289  353.87  4378.8  351.34  4396.4  349.91  4411.7  350.29  4461.1  347.97
  4600.4  342.83  4642.9  342.89  4650.6     341  4709.6  339.12  4758.4  336.46
  4789.1  336.07  4880.6  332.58  4971.2  329.22  4992.8  328.05  4997.3  326.95
  5000.1  326.45  5003.3  326.95  5035.8  328.95  5058.1  328.08  5277.6  327.64
  5358.5   330.1  5404.5  330.69  5439.4  330.05  5447.6  330.39  5453.4   332.1
    5571  335.94  5688.7  343.46  5704.5  343.58    5726   345.6  5753.7  345.95
#Mann= 6 ,-1 , 0
    4289     .05       0  4378.8      .1       0  4461.1     .05       0
  4880.6      .1       0  4997.3     .07       0  5003.3      .1       0
Bank Sta=4971.2,5035.8
XS Rating Curve= 0 ,0
Exp/Cntr=0.3,0.1

Type RM Length L Ch R = 1 ,16913   ,417,417,417
BEGIN DESCRIPTION:
UNT001 IN SPCR 28.0
END DESCRIPTION:
XS GIS Cut Line= 3
      2195687.72     13266896.86      2196337.72     13266096.85
      2196437.71     13265846.89
#Sta/Elev= 30
  3953.1  347.39  3995.5  344.62  4030.7  344.71  4060.9  342.77  4131.3  341.08
  4137.7  341.78  4159.3  338.94    4216  337.86  4223.7  338.83  4343.9  333.94
  4401.3  333.19  4521.3  328.75  4681.9  327.31  4806.1  325.83    4828  327.16
  4910.2  326.11  4927.1  325.35  4930.6  323.47  4933.3  322.97  4936.6  323.47
  4944.5  324.01  4955.9  325.35  4976.7  325.36  5005.4  324.12  5016.2  326.23
    5101   331.1  5113.1  330.72  5214.1  336.62  5238.3  339.03  5253.1  338.95
#Mann= 8 ,-1 , 0
  3953.1     .05       0  4060.9      .1       0  4681.9     .05       0
  4806.1      .1       0  4910.2     .05       0  4930.6     .07       0
  4936.6     .05       0  4944.5      .1       0
Bank Sta=4976.7,5016.2
XS Rating Curve= 0 ,0
Exp/Cntr=0.3,0.1

Type RM Length L Ch R = 1 ,16496   ,473,473,473
BEGIN DESCRIPTION:
UNT001 IN SPCR 27.0
END DESCRIPTION:
XS GIS Cut Line= 3
      2195787.69     13266896.87      2196587.72     13266396.85
      2196887.71     13266046.86
#Sta/Elev= 30
  4034.1  343.34  4230.5  335.71  4603.9  327.93  4708.1  326.06  4854.9  325.15
  4883.2  325.63  4969.9   323.8  5002.5  322.24  5005.3  321.74  5008.5  322.24
  5013.2  323.31  5027.5  323.66  5076.9  325.48  5097.7   327.4  5119.7  326.51
  5148.2  327.62  5154.8  328.96  5161.9  327.81  5169.1  328.81  5175.6  328.22
  5202.6  330.92  5211.9  330.32    5247   332.5  5261.3  332.41  5267.8  333.95
  5275.5  333.18  5289.8  333.72    5382  339.81  5388.6   341.3  5438.5  343.45
#Mann= 6 ,-1 , 0
  4034.1      .1       0  4603.9     .05       0  4854.9      .1       0
  5002.5     .07       0  5008.5      .1       0  5202.6     .05       0
Bank Sta=4969.9,5027.5
XS Rating Curve= 0 ,0
Exp/Cntr=0.3,0.1

Type RM Length L Ch R = 1 ,16023   ,597,597,597
BEGIN DESCRIPTION:
UNT001 IN SPCR 26.0
END DESCRIPTION:
XS GIS Cut Line= 3
      2195937.69     13266996.86      2196737.72     13266796.85
      2196987.72     13266246.86
#Sta/Elev= 30
  4196.1  337.74  4214.2  337.76  4255.4  335.43  4260.6  335.98  4278.6  334.75
  4301.8  334.64  4379.1  331.78  4515.7  328.35    4646  326.27  4732.1     327
  4818.9  325.22  4920.3  322.89  4943.8   321.9  4989.8  321.04  4994.6  320.17
  4997.3  319.67  5000.6  320.17  5018.2  322.83  5075.7  321.81  5104.2  322.88
  5109.7  323.75  5150.4  323.69  5178.9  324.75  5196.5  323.95  5276.7  325.24
  5482.1  332.02  5489.8  333.18    5526  333.52    5591  337.16  5624.9  338.17
#Mann= 7 ,-1 , 0
  4196.1      .1       0    4646     .05       0  4818.9     .08       0
  4943.8      .1       0  4994.6     .07       0  5000.6      .1       0
    5591     .05       0
Bank Sta=4920.3,5018.2
XS Rating Curve= 0 ,0
Exp/Cntr=0.3,0.1

Type RM Length L Ch R = 1 ,15426   ,704,704,704
BEGIN DESCRIPTION:
UNT001 IN SPCR 24.0
END DESCRIPTION:
XS GIS Cut Line= 4
      2196627.47     13267755.34      2196946.47     13267542.67
      2197181.93      13266859.1      2197204.67     13266320.86
#Sta/Elev= 30
  4258.2  333.03  4474.8  331.82  4700.6  332.97  4806.4  329.92  4850.4     327
  4869.9  325.26  4906.6  324.26  4912.2  322.44  4932.6  320.54  4969.1  320.08
  4975.6  319.11  4985.1  319.83  4986.2  319.91    4992  316.94  4994.8  316.44
    4998  316.94  5007.3  319.46  5017.9  319.82  5031.5  319.68  5081.4  322.23
  5338.4  321.37    5577  324.41    5587  323.89  5621.2  324.71  5627.1  325.77
  5663.4  325.29  5787.2  327.22  5837.2  329.08  5854.7  330.84  5903.3  332.17
#Mann= 6 ,-1 , 0
  4258.2      .1       0  4850.4     .08       0  4985.1      .1       0
    4992     .07       0    4998      .1       0  5663.4     .05       0
Bank Sta=4986.2,5017.9
XS Rating Curve= 0 ,0
Exp/Cntr=0.3,0.1

Type RM Length L Ch R = 1 ,14722   ,658,658,658
BEGIN DESCRIPTION:
Mapping XS e9afc3c6
END DESCRIPTION:
XS GIS Cut Line= 4
      2197538.15     13268101.46      2197798.56     13267736.88
      2197659.67     13266625.77      2197156.21      13266035.5
#Sta/Elev= 30
  3913.4  326.69  4025.1  325.85  4353.4  318.96  4733.6  318.56  4833.5  319.17
  4885.5   318.5  4933.4  320.01  4966.1  317.73  4983.3   315.9    4986   315.4
  4989.3   315.9  5006.4  317.42  5187.8  317.85  5429.7  322.06  5531.9  320.89
  5567.1   322.9  5573.6  321.44  5582.6  321.62    5723   321.9  5751.5  322.73
  5772.4  326.28  5786.7   326.3  5794.4  324.34  5815.2  324.17    5950  328.05
    5966  328.76  6216.5  337.13  6241.2  337.25  6247.8  338.76    6257  338.08
#Mann= 11 ,-1 , 0
  3913.4      .1       0  4025.1     .05       0  4733.6     .08       0
  4833.5     .05       0  4933.4      .1       0  4983.3     .07       0
  4989.3      .1       0  5582.6     .05       0    5950      .1       0
    5966     .05       0  6216.5      .1       0
Bank Sta=4966.1,5006.4
XS Rating Curve= 0 ,0
Exp/Cntr=0.3,0.1

Type RM Length L Ch R = 1 ,14064   ,860,860,860
BEGIN DESCRIPTION:
Mapping XS 34e0ca9e
END DESCRIPTION:
XS GIS Cut Line= 3
       2197729.1     13267979.96      2198076.34     13267511.19
      2198466.96      13265332.4
#Sta/Elev= 30
  3582.8  323.57  3798.2  318.71    3977  317.29  4700.5  316.92  4922.4  317.75
  4973.2  314.63  4989.1  312.26  4991.8  311.76  4995.1  312.26    5024  314.48
  5145.9  316.24    5255  314.25  5298.3  313.72  5349.1  317.27  5494.6  318.12
  5559.9  315.81  5625.8  318.43  5672.4   317.1  5684.3   319.4  5714.8  317.62
  5731.2  320.42  5775.8  321.42  5784.9  318.75    5790  321.87  5826.6  321.91
  5848.8   319.4  5867.2  323.33  5902.6  325.06  6009.4  326.66  6379.7  340.12
#Mann= 7 ,-1 , 0
  3582.8     .05       0  4700.5      .1       0  4989.1     .07       0
  4995.1      .1       0    5255     .08       0  5494.6     .05       0
  5625.8      .1       0
#XS Ineff= 1 ,-1
 5531.91 5622.28   318.1
Permanent Ineff=
       F
Bank Sta=4973.2,5024
XS Rating Curve= 0 ,0
Exp/Cntr=0.3,0.1

Type RM Length L Ch R = 1 ,13204   ,698,698,698
BEGIN DESCRIPTION:
Mapping XS 138de81a
END DESCRIPTION:
XS GIS Cut Line= 3
      2197824.62     13267962.55      2199282.93     13266139.66
      2199248.21      13265592.8
#Sta/Elev= 30
  3100.8  321.04  3256.6  318.41  3498.3  316.79  3946.5  316.58  4068.2  314.48
  4177.5  314.63  4436.9  314.27  4508.4  315.04  4529.6  314.16  4551.6  315.32
  4645.7  314.44  4679.7  315.43  4830.3  313.69    4907  311.44  4927.8  313.75
  4935.8  312.64  4956.6  313.09  4991.8  311.42  5003.3  308.62    5006  308.12
  5009.3  308.62  5014.3  311.44  5035.1  315.87  5113.5   319.2  5198.4  321.02
  5212.8  322.64  5418.9  328.59  5440.6  329.26  5478.1  331.58  5983.2  352.69
#Mann= 9 ,-1 , 0
  3100.8     .05       0  4177.5      .1       0  4436.9     .08       0
  4645.7     .05       0  4830.3      .1       0  5003.3     .07       0
  5009.3      .1       0  5418.9     .05       0  5440.6      .1       0
Bank Sta=4991.8,5014.3
XS Rating Curve= 0 ,0
Exp/Cntr=0.3,0.1

Type RM Length L Ch R = 1 ,12506   ,456,456,456
BEGIN DESCRIPTION:
UNT001 IN SPCR 21.0
END DESCRIPTION:
XS GIS Cut Line= 4
      2197592.03     13268621.22      2198154.12      13268294.6
      2199855.45     13266578.08      2199976.76     13266441.61
#Sta/Elev= 30
  2461.4  327.77    2659  325.66  2745.6  325.88  2956.3  322.28  3110.7  319.47
  3276.4  318.57  3279.7  318.51  3487.2  318.24  3607.4  319.38  3989.3  314.13
  4045.8  314.85  4313.9  313.31  4501.9  311.42  4603.7  309.95  4827.9  312.13
  4915.6  311.95    4958  308.96  4972.1  309.35  4979.3  310.99  4997.4  306.58
  5000.2  306.08  5003.4  306.58  5014.6  309.85  5035.8  309.32  5085.3  312.25
  5106.5  311.44  5120.7  312.84  5262.1  317.04  5290.4  319.15  5710.9  337.91
#Mann= 10 ,-1 , 0
  2461.4      .1       0  2956.3     .05       0  3276.4      .1       0
  3279.7     .05       0  4313.9      .1       0  4501.9     .08       0
  4603.7     .05       0  4827.9      .1       0  4997.4     .07       0
  5003.4      .1       0
Bank Sta=4979.3,5014.6
XS Rating Curve= 0 ,0
Exp/Cntr=0.3,0.1

Type RM Length L Ch R = 1 ,12050   ,402,402,402
BEGIN DESCRIPTION:
UNT001 IN SPCR 20.0
END DESCRIPTION:
XS GIS Cut Line= 3
      2197842.68     13268773.12      2198427.54     13268507.27
      2200082.55     13267011.69
#Sta/Elev= 30
  2604.5  325.14  2851.6  321.71  3159.5  316.38  3303.1   314.9  3615.4   314.2
  3651.3  313.17  3934.5  314.61  3962.1  315.61  3969.6  314.62  4075.7  315.83
  4174.8  314.41  4610.8  309.85  4691.5   308.6  4713.1  310.15  4755.5  309.15
  4888.7  310.92  4932.1     310    4968  307.48  4988.9  308.09  4996.3  306.82
  5000.1  304.47  5002.8  303.97  5006.1  304.47  5010.5  306.98  5031.5  308.29
  5066.7  311.76    5145   310.5  5300.5  315.39  5449.2  322.98  5477.6  325.39
#Mann= 10 ,-1 , 0
  2604.5      .1       0  2851.6     .05       0  3159.5      .1       0
  3303.1     .05       0  4174.8      .1       0  4610.8     .08       0
  4755.5     .05       0  4888.7      .1       0  5000.1     .07       0
  5006.1      .1       0
Bank Sta=4988.9,5031.5
XS Rating Curve= 0 ,0
Exp/Cntr=0.3,0.1

Type RM Length L Ch R = 1 ,11648   ,583,583,583
BEGIN DESCRIPTION:
UNT001 IN SPCR 19.0
END DESCRIPTION:
XS GIS Cut Line= 4
      2197971.81     13269069.32      2198678.19     13268765.51
      2200022.54     13267535.08      2200523.27     13267034.35
#Sta/Elev= 30
  2660.7  325.24  3198.7  315.82  3331.2  315.16  3569.8  310.57  4157.5  307.74
    4292  308.58  4504.1  310.59  4688.5  307.44  4794.1  307.84  4865.5  309.74
  4893.2  309.54  4914.8  307.28  4957.3  307.43  4992.3  306.15    5012  306.05
  5017.9  305.12  5020.6  304.62  5023.9  305.12  5028.3  307.19    5035  306.73
  5049.2  310.79  5204.9  309.23  5381.8  310.38  5657.5  322.42  5777.7  329.75
  5784.8  331.35  5834.3  332.06    5905  337.58  5940.4  338.16  5960.2  340.12
#Mann= 8 ,-1 , 0
  2660.7      .1       0  3198.7     .05       0    4292      .1       0
  4794.1     .08       0  4992.3     .05       0    5012      .1       0
  5017.9     .03       0  5023.9      .1       0
Bank Sta=4957.3,5028.3
XS Rating Curve= 0 ,0
Exp/Cntr=0.3,0.1

Type RM Length L Ch R = 1 ,11065   ,421,421,421
BEGIN DESCRIPTION:
Mapping XS be6f6079
END DESCRIPTION:
XS GIS Cut Line= 3
      2199604.64      13269603.5      2199449.91     13268991.33
      2200552.92     13267222.48
#Sta/Elev= 30
  3509.7     331  4235.1  309.99  4453.8  307.17  4463.2  305.25  4499.8  308.86
  4588.8  307.96  4688.5  306.78  4746.4  304.04  4788.8  306.17  4867.3  306.44
  4971.3  305.24  4995.8  301.19  4998.6  300.69  5001.8  301.19  5014.2  302.04
  5020.1  305.31  5045.7  305.55  5056.7  307.67    5160  307.91  5335.2  308.62
    5370  308.43  5616.9   309.1  5647.1   309.4  5731.2  310.97    5842  314.23
  5845.4  314.38  5959.7   319.6  6036.9  323.24  6073.9  324.04  6225.7  331.09
#Mann= 18 ,-1 , 0
  3509.7     .05       0  4235.1      .1       0  4588.8     .05       0
  4867.3      .1       0  4995.8     .07       0  5001.8      .1       0
  5045.7     .05       0    5160     .08       0  5335.2     .05       0
    5370      .1       0  5616.9     .08       0  5647.1      .1       0
  5731.2     .08       0    5842      .1       0  5845.4     .08       0
  5959.7      .1       0  6036.9     .08       0  6073.9      .1       0
#XS Ineff= 1 ,-1
 4255.13 4503.76  308.96
Permanent Ineff=
       F
Bank Sta=4971.3,5020.1
XS Rating Curve= 0 ,0
Exp/Cntr=0.3,0.1

Type RM Length L Ch R = 1 ,10644   ,402,402,402
BEGIN DESCRIPTION:
Mapping XS 3bfd9063
END DESCRIPTION:
XS GIS Cut Line= 3
      2199969.38     13269578.15      2200083.31     13268423.72
      2200637.74     13267345.23
#Sta/Elev= 30
  3997.4  344.51  4169.5  342.19  4219.8   338.7  4370.5  332.61  4639.6  318.65
  4852.8  310.24  4903.1  307.66  4931.9  304.47  4973.4  304.28  5000.6  300.03
  5003.3  299.53  5006.6  300.03  5013.6  303.57  5023.7  304.41    5104  306.47
  5157.4  305.34  5278.8  306.57  5351.8  307.95  5446.3  306.31  5461.3  307.84
  5572.4   307.2  5850.7  310.13  6072.5  318.16  6100.3  320.58  6116.9  319.59
  6183.4   322.6  6205.6  322.26    6250  324.76  6255.8  326.17  6370.1  330.77
#Mann= 7 ,-1 , 0
  3997.4     .05       0  4931.9      .1       0  5000.6     .07       0
  5006.6      .1       0  5278.8     .08       0  5461.3     .05       0
  5572.4      .1       0
Bank Sta=4973.4,5023.7
XS Rating Curve= 0 ,0
Exp/Cntr=0.3,0.1

Type RM Length L Ch R = 1 ,10242   ,579,579,579
BEGIN DESCRIPTION:
Mapping XS e9569f0f
END DESCRIPTION:
XS GIS Cut Line= 3
      2200858.03     13269904.83      2200394.71     13268484.48
      2200652.42      13267400.6
#Sta/Elev= 30
  3679.5  328.59  3955.4  327.49  4146.8   322.7    4152  323.74  4242.5  320.48
  4247.7  321.32  4396.9  316.22  4439.1  315.82  4455.7  314.28  4694.3  307.24
  4699.6  308.14  4758.1  306.11  4795.3  306.44  4949.5  302.76  4986.7  302.91
  4999.7  298.64  5002.5  298.14  5005.7  298.64  5018.6  303.92  5044.8  304.23
  5065.8  302.82  5100.2  303.91  5160.5  304.36  5181.3  305.72  5212.7  304.57
  5265.3  305.45  5431.2   305.8  5623.3  307.86  5839.2  313.68  6287.6  329.74
#Mann= 7 ,-1 , 0
  3679.5     .05       0  4396.9      .1       0  4999.7     .07       0
  5005.7      .1       0  5100.2     .08       0  5265.3     .05       0
  5431.2      .1       0
Bank Sta=4986.7,5018.6
XS Rating Curve= 0 ,0
Exp/Cntr=0.3,0.1

Type RM Length L Ch R = 1 ,9663    ,1182,1182,1182
BEGIN DESCRIPTION:
Mapping XS 7d00d375
END DESCRIPTION:
XS GIS Cut Line= 4
      2201979.12      13270074.3      2201232.49     13269220.03
      2200714.53     13268089.95      2200775.07     13267417.26
#Sta/Elev= 30
  3268.8  319.11  3459.4  313.13  3508.8   313.3  3516.4   312.2  3636.9  310.19
    3957  308.11  4091.8  307.16  4187.1  306.71  4226.5   306.5  4331.3  305.79
  4361.3  305.56  4448.1  304.72  4471.1  306.64  4476.6  304.57  4483.9  306.45
  4689.1  302.13  4840.2  302.56  4981.6  301.63  4989.9  297.14  4996.1  296.61
  4998.8  296.11  5002.1  296.61  5033.9  302.52  5079.1  300.57  5176.9  303.96
  5463.6  306.47  5669.7  310.72  5807.8  315.66  5931.3   320.3  6321.9  332.21
#Mann= 12 ,-1 , 0
  3268.8     .08       0    3957      .1       0  4091.8     .05       0
  4187.1      .1       0  4226.5     .05       0  4331.3      .1       0
  4361.3     .05       0  4840.2      .1       0  4996.1     .07       0
  5002.1      .1       0  5807.8     .05       0  5931.3      .1       0
Bank Sta=4981.6,5033.9
XS Rating Curve= 0 ,0
Exp/Cntr=0.3,0.1

Type RM Length L Ch R = 1 ,8481    ,784,784,784
BEGIN DESCRIPTION:
Mapping XS 3cef75ba
END DESCRIPTION:
XS GIS Cut Line= 3
      2202361.88     13270299.75      2202118.83     13269236.41
      2202042.88      13267216.1
#Sta/Elev= 30
  3522.4  324.05  3803.9  317.36    4346  304.92  4608.2  302.35  4714.4   300.5
  4802.8  298.32  4872.9  299.43  4942.9  296.73    4983   297.8    4993  291.98
    5000  291.49  5002.7  290.99    5006  291.49    5013  295.85    5023  297.32
    5053  296.59  5203.1  301.31  5593.4  302.07  5733.5  306.56  5823.6   307.2
  5873.6  311.64  5893.6  310.37  6029.1  318.17    6127  323.21  6313.9  335.68
  6380.2  337.76    6444  342.95  6514.1  344.95  6544.1  347.73  6634.9  348.39
#Mann= 9 ,-1 , 0
  3522.4     .05       0  3803.9      .1       0  4608.2     .05       0
  4714.4      .1       0    5000     .07       0    5006      .1       0
  6029.1     .05       0    6127      .1       0  6380.2     .05       0
Bank Sta=4983,5023
XS Rating Curve= 0 ,0
Exp/Cntr=0.3,0.1
