HEC-RAS study ROCK QUARRY BRANCH.prj: ROCK QUARRY BRANCH Base Level Engineering

--- ROCK QUARRY BRANCH.g01 (geometry) --- (continued)

Type RM Length L Ch R = 1 ,34580   ,335,335,335
BEGIN DESCRIPTION:
Mapping XS 69c3c86b
END DESCRIPTION:
XS GIS Cut Line= 4
      2244819.97     13375917.43      2244076.04     13375654.15
      2243609.88     13375574.45      2243235.55     13375562.37
#Sta/Elev= 30
  4110.6  246.18  4395.6  237.84  4420.6   237.6  4426.5  238.51  4441.8  238.53
  4452.1   237.4    4483  236.36  4569.1  237.35  4753.1  235.01  4781.3  234.85
  4786.7  235.63  4802.5  234.62  4843.2  235.52  4899.8  235.19  4989.3  233.95
    4997  232.87  4999.8  232.37    5003  232.87  5009.6  234.06  5050.2  232.87
  5213.8  237.04  5434.9   245.4  5444.9   245.2  5451.5  246.16  5484.9  247.44
  5544.9  248.57  5594.9  251.13    5675  253.46    5735  253.93  5747.2  255.34
#Mann= 4 ,-1 , 0
  4110.6     .05       0  4753.1      .1       0    4997     .07       0
    5003      .1       0
Bank Sta=4997,5003
XS Rating Curve= 0 ,0
Exp/Cntr=0.3,0.1

Type RM Length L Ch R = 1 ,34563   ,334,334,334
BEGIN DESCRIPTION:
Mapping XS 69c3c86b
END DESCRIPTION:
XS GIS Cut Line= 4
      2244819.97     13375917.43      2244076.04     13375654.15
      2243609.88     13375574.45      2243235.55     13375562.37
#Sta/Elev= 30
  4110.6  246.18  4395.6  237.84  4420.6   237.6  4426.5  238.51  4441.8  238.53
  4452.1   237.4  4457.4  237.75    4483  236.36  4569.1  237.35  4753.1  235.01
  4781.3  234.85  4786.7  235.63  4802.5  234.62  4866.1  235.46  4938.6  234.45
  4973.4  233.73  5019.8  234.09  5047.2  232.87    5050  232.37  5053.2  232.87
  5273.9  238.92  5434.9   245.4  5444.9   245.2  5451.5  246.16  5484.9  247.44
  5544.9  248.57  5594.9  251.13    5675  253.46    5735  253.93  5747.2  255.34
#Mann= 4 ,-1 , 0
  4110.6     .05       0  4753.1      .1       0  5047.2     .07       0
  5053.2      .1       0
Bank Sta=4938.6,5019.8
XS Rating Curve= 0 ,0
Exp/Cntr=0.3,0.1

Type RM Length L Ch R = 1 ,34245   ,602,602,602
BEGIN DESCRIPTION:
ROCK QUARRY BRANCH 63.0
END DESCRIPTION:
XS GIS Cut Line= 2
      2245236.01     13375585.59      2243495.03     13375193.89
#Sta/Elev= 30
  3801.8  252.86  3957.2  249.48  4220.3  240.74  4318.8  238.17  4550.6  234.42
  4722.5  233.56  4753.3  232.49  4835.3  232.67  4917.3  231.79  4937.8  232.53
  4955.5  230.98  4978.8  231.11    4997  230.06  4999.8  229.56    5003  230.06
  5003.9   230.8  5019.8  231.69  5040.3  231.25  5069.6  232.77  5094.2  233.44
  5108.4   233.5  5132.5  233.41  5224.8  236.25  5273.8  238.66  5306.8  239.64
    5317   239.1  5365.5  241.39    5440  243.17  5457.2  244.28  5586.3  248.22
#Mann= 6 ,-1 , 0
  3801.8     .05       0    4997     .03       0    5003     .05       0
  5069.6      .1       0  5094.2     .05       0  5108.4      .1       0
Bank Sta=4997,5003
XS Rating Curve= 0 ,0
Exp/Cntr=0.3,0.1

Type RM Length L Ch R = 1 ,34229   ,602,602,602
BEGIN DESCRIPTION:
ROCK QUARRY BRANCH 63.0
END DESCRIPTION:
XS GIS Cut Line= 2
      2245236.01     13375585.59      2243495.03     13375193.89
#Sta/Elev= 30
  3801.8  252.86  3957.2  249.48  4097.3   245.4  4220.3  240.74  4318.8  238.17
  4550.6  234.42  4722.5  233.56  4753.3  232.49  4835.3  232.67  4917.3  231.79
  4937.8  232.53  4955.5  230.98  4978.8  231.11    4986  230.06  4988.8  229.56
    4992  230.06  5019.8  231.69  5040.3  231.25  5069.6  232.77  5094.2  233.44
  5108.4   233.5  5132.5  233.41  5224.8  236.25  5273.8  238.66  5306.8  239.64
    5317   239.1  5365.5  241.39    5440  243.17  5457.2  244.28  5586.3  248.22
#Mann= 6 ,-1 , 0
  3801.8     .05       0    4986     .03       0    4992     .05       0
  5069.6      .1       0  5094.2     .05       0  5108.4      .1       0
Bank Sta=4937.8,5069.6
XS Rating Curve= 0 ,0
Exp/Cntr=0.3,0.1

Type RM Length L Ch R = 1 ,33643   ,174,174,174
BEGIN DESCRIPTION:
ROCK QUARRY BRANCH 62.0
END DESCRIPTION:
XS GIS Cut Line= 4
      2245127.01     13375166.13       2244550.6     13374853.62
      2244342.27     13374832.79       2243628.5     13374992.17
#Sta/Elev= 30
  4199.7  248.15  4250.4  246.21  4310.3  245.25  4337.8  243.07  4419.6  240.33
  4551.5  237.67  4722.2  232.98  4824.5  231.19  4873.2  231.19  4898.5  226.95
  4908.5   224.1  4928.6   221.5    4997  219.27  4999.8  218.77    5003  219.27
  5049.2  220.17  5069.6  221.35  5089.9  223.58  5105.8  227.81  5110.9  228.04
  5120.6  230.14  5141.1  232.04  5262.8  232.37  5381.8  234.11  5565.8  238.16
    5592  239.13  5602.2  240.55    5633  240.54  5755.9  245.57  5796.1  245.95
#Mann= 4 ,-1 , 0
  4199.7     .05       0    4997     .03       0    5003     .05       0
  5262.8      .1       0
Bank Sta=4997,5003
XS Rating Curve= 0 ,0
Exp/Cntr=0.3,0.1

Type RM Length L Ch R = 1 ,33627   ,174,174,174
BEGIN DESCRIPTION:
ROCK QUARRY BRANCH 62.0
END DESCRIPTION:
XS GIS Cut Line= 4
      2245127.01     13375166.13       2244550.6     13374853.62
      2244342.27     13374832.79       2243628.5     13374992.17
#Sta/Elev= 30
  4199.7  248.15  4250.4  246.21  4310.3  245.25  4337.8  243.07  4419.6  240.33
  4551.5  237.67  4722.2  232.98  4824.5  231.19  4873.2  231.19  4898.5  226.95
  4908.5   224.1  4928.6   221.5  4958.8  220.01    5006  219.27  5008.8  218.77
    5012  219.27  5069.6  221.35  5089.9  223.58  5105.8  227.81  5130.9  231.42
  5161.6  232.29  5171.9  231.66  5262.8  232.37  5381.8  234.11  5565.8  238.16
    5592  239.13  5602.2  240.55    5633  240.54  5755.9  245.57  5796.1  245.95
#Mann= 4 ,-1 , 0
  4199.7     .05       0    5006     .03       0    5012     .05       0
  5262.8      .1       0
Bank Sta=4873.2,5130.9
XS Rating Curve= 0 ,0
Exp/Cntr=0.3,0.1

Type RM Length L Ch R = 1 ,33469   ,113,113,113
BEGIN DESCRIPTION:
Mapping XS 2e796d4d
END DESCRIPTION:
XS GIS Cut Line= 4
      2245224.22     13375055.01      2244578.38     13374728.62
      2244432.55      13374693.9      2243592.48     13374888.29
#Sta/Elev= 30
  4211.5  250.22  4332.9   246.1  4371.9  243.77  4521.3   240.3  4594.8  237.33
  4667.2  236.85  4745.2  233.34  4839.9  231.23  4856.6  233.24  4862.2  232.89
  4868.6  234.42  4878.9  235.08  4884.5  233.98  4901.2  235.96  4962.9  234.95
  4968.1  235.85  4987.2  235.13    4997  231.23  4999.8  230.73    5003  231.23
  5005.1  234.21  5010.2  235.77  5059.2  236.31  5299.1  235.75  5335.2  234.23
  5341.8  233.28  5346.9  235.43  5459.5  233.63  5565.6  235.51  5947.3  247.34
#Mann= 4 ,-1 , 0
  4211.5     .05       0    4997     .03       0    5003     .05       0
  5335.2      .1       0
Bank Sta=4997,5003
XS Rating Curve= 0 ,0
Exp/Cntr=0.3,0.1

Type RM Length L Ch R = 1 ,33453   ,114,114,114
BEGIN DESCRIPTION:
Mapping XS 2e796d4d
END DESCRIPTION:
XS GIS Cut Line= 4
      2245224.22     13375055.01      2244578.38     13374728.62
      2244432.55      13374693.9      2243592.48     13374888.29
#Sta/Elev= 30
  4211.5  250.22  4332.9   246.1  4371.9  243.77  4521.3   240.3  4594.8  237.33
  4622.7  237.88  4667.2  236.85  4745.2  233.34  4795.4  232.95  4836.9  231.23
  4839.7  230.73  4842.9  231.23  4846.2   232.4  4862.2  232.89  4868.6  234.42
  4878.9  235.08  4884.5  233.98  4901.2  235.96  4962.9  234.95  4968.1  235.85
  5005.1  234.21  5010.2  235.77  5192.6  236.35  5315.8  235.53  5335.2  234.23
  5341.8  233.28  5346.9  235.43  5459.5  233.63  5565.6  235.51  5947.3  247.34
#Mann= 4 ,-1 , 0
  4211.5     .05       0  4836.9     .03       0  4842.9     .05       0
  5335.2      .1       0
Bank Sta=4968.1,5010.2
XS Rating Curve= 0 ,0
Exp/Cntr=0.3,0.1

Type RM Length L Ch R = 1 ,33356   ,381,381,381
BEGIN DESCRIPTION:
ROCK QUARRY BRANCH 61.0
END DESCRIPTION:
XS GIS Cut Line= 3
      2245187.67     13374696.85      2244537.72     13374596.85
      2243437.75     13374796.85
#Sta/Elev= 30
  4322.5  247.49  4419.8  243.46  4483.1  241.36  4494.5  241.54  4646.2  236.14
  4676.6  235.84  4727.2  233.75  4877.7  229.93  4959.9  229.09    4997  227.66
  4999.8  227.16    5003  227.66  5011.9  228.77  5051.2  227.66  5081.7  229.91
  5123.7  230.59  5295.2  231.29  5303.9  230.73  5559.4  235.58  5579.8  236.83
  5589.9  236.41  5661.1  238.79  5691.6  239.14    5731  241.23    5736  240.46
    5783  242.06  5789.4  242.88  5847.8  243.93  5945.7  247.25  6098.1  250.23
#Mann= 4 ,-1 , 0
  4322.5     .05       0    4997     .03       0    5003     .05       0
  5303.9      .1       0
Bank Sta=4997,5003
XS Rating Curve= 0 ,0
Exp/Cntr=0.3,0.1

Type RM Length L Ch R = 1 ,33339   ,380,380,380
BEGIN DESCRIPTION:
ROCK QUARRY BRANCH 61.0
END DESCRIPTION:
XS GIS Cut Line= 3
      2245187.67     13374696.85      2244537.72     13374596.85
      2243437.75     13374796.85
#Sta/Elev= 30
  4322.5  247.49  4419.8  243.46  4483.1  241.36  4494.5  241.54  4646.2  236.14
  4676.6  235.84  4727.2  233.75  4877.7  229.93  4959.9  229.09  4977.6  227.96
  5011.9  228.77  5048.2  227.66    5051  227.16  5054.2  227.66  5071.6  229.22
  5132.6  230.67  5295.2  231.29  5303.9  230.73  5559.4  235.58  5579.8  236.83
  5589.9  236.41  5661.1  238.79  5691.6  239.14    5731  241.23    5736  240.46
    5783  242.06  5789.4  242.88  5847.8  243.93  5945.7  247.25  6098.1  250.23
#Mann= 4 ,-1 , 0
  4322.5     .05       0  5048.2     .03       0  5054.2     .05       0
  5303.9      .1       0
Bank Sta=4959.9,5071.6
XS Rating Curve= 0 ,0
Exp/Cntr=0.3,0.1

Type RM Length L Ch R = 1 ,32975   ,391,391,391
BEGIN DESCRIPTION:
ROCK QUARRY BRANCH 60.0
END DESCRIPTION:
XS GIS Cut Line= 3
      2245137.68     13374346.85      2244387.72     13374246.85
      2243587.72     13374546.86
#Sta/Elev= 30
  4288.3  244.17  4389.1  241.19  4409.3  241.49  4419.4  240.46  4460.3  238.87
  4522.7  237.41  4611.1  235.77  4692.2  233.27  4778.8  231.27  4843.1  230.82
    4852  229.93    4857  230.49  4913.7  228.48  4984.4  227.15    4997  226.19
  4999.8  225.69    5003  226.19  5024.7  227.75  5034.8   227.3    5060  228.08
  5291.4  229.74  5487.2  234.42  5567.3  236.98  5597.6  238.76  5610.9  238.54
  5652.8   240.3  5688.4  240.63  5713.3   242.1  5743.5  242.12  5899.3  245.87
#Mann= 6 ,-1 , 0
  4288.3     .05       0  4460.3      .1       0  4522.7     .05       0
  4692.2      .1       0    4997     .07       0    5003      .1       0
Bank Sta=4997,5003
XS Rating Curve= 0 ,0
Exp/Cntr=0.3,0.1

Type RM Length L Ch R = 1 ,32959   ,391,391,391
BEGIN DESCRIPTION:
ROCK QUARRY BRANCH 60.0
END DESCRIPTION:
XS GIS Cut Line= 3
      2245137.68     13374346.85      2244387.72     13374246.85
      2243587.72     13374546.86
#Sta/Elev= 30
  4288.3  244.17  4389.1  241.19  4409.3  241.49  4419.4  240.46  4460.3  238.87
  4522.7  237.41  4611.1  235.77  4692.2  233.27  4778.8  231.27  4843.1  230.82
    4852  229.93    4857  230.49    4944  227.96  5000.3  226.19    5003  225.69
  5006.3  226.19  5024.7  227.75  5034.8   227.3    5060  228.08  5291.4  229.74
  5487.2  234.42  5567.3  236.98  5597.6  238.76  5610.9  238.54  5652.8   240.3
  5688.4  240.63  5713.3   242.1  5743.5  242.12  5884.2  245.99  5899.3  245.87
#Mann= 6 ,-1 , 0
  4288.3     .05       0  4460.3      .1       0  4522.7     .05       0
  4692.2      .1       0  5000.3     .07       0  5006.3      .1       0
Bank Sta=4944,5024.7
XS Rating Curve= 0 ,0
Exp/Cntr=0.3,0.1

Type RM Length L Ch R = 1 ,32584   ,552,552,552
BEGIN DESCRIPTION:
ROCK QUARRY BRANCH 59.0
END DESCRIPTION:
XS GIS Cut Line= 3
      2244902.16     13373790.47      2244611.36     13373794.81
       2243536.6     13374232.52
#Sta/Elev= 30
  4248.1  240.16  4679.3   231.8  4718.8  231.74  4737.2  230.73    4856  228.88
  4951.5  226.09    4981  225.99    4997  224.62  4999.8  224.12    5003  224.62
  5010.4   225.8  5017.9  225.91  5058.5  225.26  5063.9  226.28  5082.6   225.9
    5088  226.54  5093.5  225.88  5104.3  225.93  5125.9  227.84    5171  228.88
  5179.9  229.61  5266.3  230.63  5433.1  237.02  5510.6  238.65  5557.8  240.28
  5564.2  241.03  5593.6   240.9  5665.8   242.6  5671.2  243.44  5699.4  244.26
#Mann= 4 ,-1 , 0
  4248.1     .05       0  4679.3      .1       0    4997     .07       0
    5003      .1       0
Bank Sta=4997,5003
XS Rating Curve= 0 ,0
Exp/Cntr=0.3,0.1

Type RM Length L Ch R = 1 ,32568   ,553,553,553
BEGIN DESCRIPTION:
ROCK QUARRY BRANCH 59.0
END DESCRIPTION:
XS GIS Cut Line= 3
      2244902.16     13373790.47      2244611.36     13373794.81
       2243536.6     13374232.52
#Sta/Elev= 30
  4248.1  240.16  4679.3   231.8  4718.8  231.74  4737.2  230.73  4772.4  230.57
  4903.4  227.78  4951.5  226.09    4981  225.99  4993.4  224.62  4996.1  224.12
  4999.4  224.62  5017.9  225.91  5058.5  225.26  5063.9  226.28  5082.6   225.9
    5088  226.54  5093.5  225.88  5104.3  225.93  5125.9  227.84    5171  228.88
  5179.9  229.61  5266.3  230.63  5433.1  237.02  5510.6  238.65  5557.8  240.28
  5564.2  241.03  5593.6   240.9  5665.8   242.6  5671.2  243.44  5699.4  244.26
#Mann= 4 ,-1 , 0
  4248.1     .05       0  4679.3      .1       0  4993.4     .07       0
  4999.4      .1       0
Bank Sta=4981,5017.9
XS Rating Curve= 0 ,0
Exp/Cntr=0.3,0.1

Type RM Length L Ch R = 1 ,32032   ,499,499,499
BEGIN DESCRIPTION:
ROCK QUARRY BRANCH 58.0
END DESCRIPTION:
XS GIS Cut Line= 2
      2244767.62     13373499.68      2243443.83     13373517.04
#Sta/Elev= 30
  4227.2  237.62    4653  230.54  4747.1  229.23  4767.1  228.39  4787.1  228.81
  4817.1  227.71  4927.2  225.73  4947.2  224.55  4987.2  223.71    4997  222.57
  4999.8  222.07    5003  222.57  5007.2  224.14  5017.2  223.44  5027.2  224.14
  5107.2   225.6  5137.2  227.41  5154.1  227.42  5167.2  228.93  5177.2   228.4
  5227.2  229.71  5237.2  230.56  5257.2  230.58  5267.2  231.66  5277.2  231.27
  5307.2  232.68  5347.2  233.34  5367.2  234.43  5543.3  239.96  5551.1  240.16
#Mann= 5 ,-1 , 0
  4227.2     .05       0    4653      .1       0    4997     .07       0
    5003      .1       0  5543.3     .05       0
Bank Sta=4997,5003
XS Rating Curve= 0 ,0
Exp/Cntr=0.3,0.1

Type RM Length L Ch R = 1 ,32015   ,499,499,499
BEGIN DESCRIPTION:
ROCK QUARRY BRANCH 58.0
END DESCRIPTION:
XS GIS Cut Line= 2
      2244767.62     13373499.68      2243443.83     13373517.04
#Sta/Elev= 30
  4227.2  237.62    4653  230.54  4747.1  229.23  4767.1  228.39  4787.1  228.81
  4957.2  224.65  4987.2  223.71  4994.2  222.57  4996.9  222.07  5000.2  222.57
  5007.2  224.14  5017.2  223.44  5027.2  224.14  5057.2  224.29  5107.2   225.6
  5137.2  227.41  5154.1  227.42  5167.2  228.93  5177.2   228.4  5227.2  229.71
  5237.2  230.56  5257.2  230.58  5267.2  231.66  5277.2  231.27  5307.2  232.68
  5347.2  233.34  5367.2  234.43  5397.2  234.98  5543.3  239.96  5551.1  240.16
#Mann= 5 ,-1 , 0
  4227.2     .05       0    4653      .1       0  4994.2     .07       0
  5000.2      .1       0  5543.3     .05       0
Bank Sta=4957.2,5007.2
XS Rating Curve= 0 ,0
Exp/Cntr=0.3,0.1

Type RM Length L Ch R = 1 ,31533   ,438,438,438
BEGIN DESCRIPTION:
ROCK QUARRY BRANCH 57.0
END DESCRIPTION:
XS GIS Cut Line= 3
      2244787.75     13373146.86      2243987.72     13373046.85
      2243487.69     13373196.86
#Sta/Elev= 30
  4215.2  238.12    4765  228.21    4830  227.27    4898  225.65  4950.9  223.95
  4978.6  222.62  4991.2   222.5    4997  221.74  4999.8  221.24    5003  221.74
  5011.4  223.17  5024.1  222.63  5031.9  221.74    5038  222.54  5104.1  223.64
  5188.5   226.7  5216.6  227.21  5285.1  229.93  5356.4  231.16  5376.4  232.08
  5384.3  233.08  5397.3  233.76  5422.5  234.66  5449.5  235.07  5460.8  236.08
  5493.9  237.22  5512.2  238.52  5526.9  238.34    5533  239.28  5543.5  239.72
#Mann= 5 ,-1 , 0
  4215.2     .05       0    4765      .1       0    4997     .07       0
    5003      .1       0  5216.6     .05       0
Bank Sta=4997,5003
XS Rating Curve= 0 ,0
Exp/Cntr=0.3,0.1

Type RM Length L Ch R = 1 ,31516   ,437,437,437
BEGIN DESCRIPTION:
ROCK QUARRY BRANCH 57.0
END DESCRIPTION:
XS GIS Cut Line= 3
      2244787.75     13373146.86      2243987.72     13373046.85
      2243487.69     13373196.86
#Sta/Elev= 30
  4215.2  238.12    4765  228.21    4830  227.27  4890.4  225.86    4961  223.43
  5001.3  222.05  5011.4  223.17  5024.1  222.63  5028.9  221.74  5031.6  221.24
  5034.9  221.74    5038  222.54  5063.2  222.82    5071  223.26  5104.1  223.64
  5188.5   226.7  5216.6  227.21  5285.1  229.93  5356.4  231.16  5376.4  232.08
  5384.3  233.08  5397.3  233.76  5422.5  234.66  5449.5  235.07  5460.8  236.08
  5493.9  237.22  5512.2  238.52  5526.9  238.34    5533  239.28  5543.5  239.72
#Mann= 5 ,-1 , 0
  4215.2     .05       0    4765      .1       0  5028.9     .07       0
  5034.9      .1       0  5216.6     .05       0
Bank Sta=4961,5071
XS Rating Curve= 0 ,0
Exp/Cntr=0.3,0.1

Type RM Length L Ch R = 1 ,31095   ,438,438,438
BEGIN DESCRIPTION:
ROCK QUARRY BRANCH 56.0
END DESCRIPTION:
XS GIS Cut Line= 3
      2244787.74     13372596.85      2243987.72     13372646.85
      2243287.71     13372446.85
#Sta/Elev= 30
    4175  237.34  4265.2  235.32  4305.3  233.49  4375.4   232.3    4413  230.37
  4513.8  228.47  4645.9  225.93  4738.6  225.44  4776.2  224.72  4796.2  223.38
  4816.3  223.97  4936.5  221.56    4987  221.35    4997  220.21  4999.8  219.71
    5003  220.21  5059.8  222.61  5211.9   226.8  5226.2  226.36  5289.9  227.51
    5299  228.91  5318.5  229.56  5330.2  228.45    5351  229.54  5362.7  229.21
  5382.2  231.31  5413.4  231.53  5449.1  233.04  5621.4   239.1  5704.6  240.88
#Mann= 5 ,-1 , 0
    4175     .05       0  4513.8      .1       0    4997     .07       0
    5003      .1       0  5449.1     .05       0
Bank Sta=4997,5003
XS Rating Curve= 0 ,0
Exp/Cntr=0.3,0.1

Type RM Length L Ch R = 1 ,31079   ,438,438,438
BEGIN DESCRIPTION:
ROCK QUARRY BRANCH 56.0
END DESCRIPTION:
XS GIS Cut Line= 3
      2244787.74     13372596.85      2243987.72     13372646.85
      2243287.71     13372446.85
#Sta/Elev= 30
    4175  237.34  4265.2  235.32  4305.3  233.49  4375.4   232.3    4413  230.37
  4513.8  228.47  4645.9  225.93  4738.6  225.44  4776.2  224.72  4796.2  223.38
  4816.3  223.97  4936.5  221.56    4987  221.35  4995.7  220.21  4998.4  219.71
  5001.7  220.21  5027.3  221.41  5211.9   226.8  5226.2  226.36  5289.9  227.51
    5299  228.91  5318.5  229.56  5330.2  228.45    5351  229.54  5362.7  229.21
  5382.2  231.31  5413.4  231.53  5449.1  233.04  5621.4   239.1  5704.6  240.88
#Mann= 5 ,-1 , 0
    4175     .05       0  4513.8      .1       0  4995.7     .07       0
  5001.7      .1       0  5449.1     .05       0
Bank Sta=4987,5027.3
XS Rating Curve= 0 ,0
Exp/Cntr=0.3,0.1

Type RM Length L Ch R = 1 ,30657   ,573,573,573
BEGIN DESCRIPTION:
ROCK QUARRY BRANCH 55.0
END DESCRIPTION:
XS GIS Cut Line= 3
      2244887.69     13372096.86      2244087.72     13372246.85
      2243287.69     13372296.86
#Sta/Elev= 30
  4186.3  240.93  4308.4  235.42  4322.8  236.04  4338.9  234.69  4440.6  231.19
  4543.2   229.3  4613.6  226.58  4734.4  223.89  4821.3  222.28  4921.8  220.69
    4997  219.07  4999.8  218.57    5003  219.07  5010.2  220.18  5187.5   223.5
  5340.9  226.56  5360.9  232.38  5370.9  233.09    5381  233.37  5395.6  229.75
  5398.5  229.14  5403.5  230.22    5411  228.36    5421  228.45  5461.1  230.88
  5563.8  233.34  5581.3  234.88  5651.5  235.93  5771.7   241.3  5801.8  241.66
#Mann= 8 ,-1 , 0
  4186.3      .1       0  4734.4     .12       0  4821.3      .1       0
  4921.8     .12       0    4997     .07       0    5003     .12       0
  5187.5      .1       0  5395.6     .05       0
Bank Sta=4997,5003
XS Rating Curve= 0 ,0
Exp/Cntr=0.3,0.1

Type RM Length L Ch R = 1 ,30641   ,573,573,573
BEGIN DESCRIPTION:
ROCK QUARRY BRANCH 55.0
END DESCRIPTION:
XS GIS Cut Line= 3
      2244887.69     13372096.86      2244087.72     13372246.85
      2243287.69     13372296.86
#Sta/Elev= 30
  4186.3  240.93  4308.4  235.42  4322.8  236.04  4338.9  234.69  4440.6  231.19
  4543.2   229.3  4734.4  223.89  4821.3  222.28  4921.4   220.7  4921.8  220.69
    4987  219.07  4989.8  218.57    4993  219.07  5040.3  220.76  5187.5   223.5
  5340.9  226.56  5360.9  232.38  5370.9  233.09    5381  233.37  5395.6  229.75
  5398.5  229.14  5403.5  230.22    5411  228.36    5421  228.45  5461.1  230.88
  5563.8  233.34  5581.3  234.88  5651.5  235.93  5771.7   241.3  5801.8  241.66
#Mann= 8 ,-1 , 0
  4186.3      .1       0  4734.4     .12       0  4821.3      .1       0
  4921.8     .12       0    4987     .07       0    4993     .12       0
  5187.5      .1       0  5395.6     .05       0
Bank Sta=4921.4,5040.3
XS Rating Curve= 0 ,0
Exp/Cntr=0.3,0.1

Type RM Length L Ch R = 1 ,30084   ,390,390,390
BEGIN DESCRIPTION:
ROCK QUARRY BRANCH 54.0
END DESCRIPTION:
XS GIS Cut Line= 4
      2244953.34     13371846.67      2244585.33      13371756.4
      2243870.05     13371714.73      2243383.93     13371916.12
#Sta/Elev= 30
    4273  241.17  4364.4  238.65  4412.6  237.94  4423.6   236.5  4474.4  235.21
  4484.7  232.77  4501.6  232.45  4506.8  234.05  4515.6  234.21  4536.2   233.6
  4709.6  226.19  4749.7  223.36  4889.9  220.02  4970.1  219.34  4990.1  220.16
    4997  219.25  4999.8  218.75    5003  219.25  5019.5  219.78  5053.5   220.2
  5090.3  220.41  5120.3  222.71  5280.6  223.54  5330.7  226.21  5536.7  228.19
  5800.9  233.25  5814.7  233.72  5825.6  232.68  5894.3  234.91  5894.6  234.91
#Mann= 9 ,-1 , 0
    4273     .05       0  4364.4      .1       0    4997     .07       0
    5003      .1       0  5019.5     .12       0  5053.5      .1       0
  5536.7     .05       0  5800.9      .1       0  5894.3     .05       0
Bank Sta=4997,5003
XS Rating Curve= 0 ,0
Exp/Cntr=0.3,0.1

Type RM Length L Ch R = 1 ,30068   ,391,391,391
BEGIN DESCRIPTION:
ROCK QUARRY BRANCH 54.0
END DESCRIPTION:
XS GIS Cut Line= 4
      2244953.34     13371846.67      2244585.33      13371756.4
      2243870.05     13371714.73      2243383.93     13371916.12
#Sta/Elev= 30
    4273  241.17  4364.4  238.65  4412.6  237.94  4423.6   236.5  4474.4  235.21
  4484.7  232.77  4501.6  232.45  4506.8  234.05  4515.6  234.21  4536.2   233.6
  4709.6  226.19  4749.7  223.36    4920  219.57  4990.1  220.16  5007.1  219.25
  5009.9  218.75  5013.1  219.25  5019.5  219.76  5053.5   220.2  5069.6  220.69
  5090.3  220.41  5120.3  222.71  5280.6  223.54  5330.7  226.21  5536.7  228.19
  5800.9  233.25  5814.7  233.72  5825.6  232.68  5894.3  234.91  5894.6  234.91
#Mann= 9 ,-1 , 0
    4273     .05       0  4364.4      .1       0  5007.1     .07       0
  5013.1      .1       0  5019.5     .12       0  5053.5      .1       0
  5536.7     .05       0  5800.9      .1       0  5894.3     .05       0
Bank Sta=4990.1,5069.6
XS Rating Curve= 0 ,0
Exp/Cntr=0.3,0.1

Type RM Length L Ch R = 1 ,29694   ,444,444,444
BEGIN DESCRIPTION:
ROCK QUARRY BRANCH 53.0
END DESCRIPTION:
XS GIS Cut Line= 3
      2244737.76     13371396.85      2244337.72     13371396.85
      2243537.71     13371546.86
#Sta/Elev= 30
  4591.8  231.34  4621.8  229.68  4631.8  229.37  4641.8  229.64  4651.8  228.87
  4681.8  228.12  4711.8  226.55  4731.8  226.04  4751.8  224.82  4781.8  223.83
  4801.8  223.66  4841.8  221.22  4872.2  220.38  4901.8  218.33  4941.8  217.04
    4997  216.06  4999.8  215.56    5003  216.06  5018.1  216.99  5042.8  217.58
  5128.3   219.9  5134.3  220.48  5144.5  220.29  5317.4  223.79  5551.4  227.13
    5582  227.95  5616.7  228.18  5734.6  230.39  5765.1  230.55  5805.8  231.69
#Mann= 5 ,-1 , 0
  4591.8      .1       0  4872.2     .12       0    4997     .07       0
    5003     .12       0  5042.8     .05       0
Bank Sta=4997,5003
XS Rating Curve= 0 ,0
Exp/Cntr=0.3,0.1

Type RM Length L Ch R = 1 ,29677   ,444,444,444
BEGIN DESCRIPTION:
ROCK QUARRY BRANCH 53.0
END DESCRIPTION:
XS GIS Cut Line= 3
      2244737.76     13371396.85      2244337.72     13371396.85
      2243537.71     13371546.86
#Sta/Elev= 30
  4591.8  231.34  4621.8  229.68  4631.8  229.37  4641.8  229.64  4651.8  228.87
  4681.8  228.12  4711.8  226.55  4731.8  226.04  4751.8  224.82  4781.8  223.83
  4801.8  223.66  4841.8  221.22  4872.2  220.38  4901.8  218.33  4941.8  217.04
    4999  216.06  5001.8  215.56    5005  216.06  5018.1  216.99  5042.8  217.58
  5128.3   219.9  5134.3  220.48  5144.5  220.29  5317.4  223.79  5551.4  227.13
    5582  227.95  5616.7  228.18  5734.6  230.39  5765.1  230.55  5805.8  231.69
#Mann= 5 ,-1 , 0
  4591.8      .1       0  4872.2     .12       0    4999     .07       0
    5005     .12       0  5042.8     .05       0
Bank Sta=4941.8,5018.1
XS Rating Curve= 0 ,0
Exp/Cntr=0.3,0.1

Type RM Length L Ch R = 1 ,29250   ,495,495,495
BEGIN DESCRIPTION:
ROCK QUARRY BRANCH 52.0
END DESCRIPTION:
XS GIS Cut Line= 3
      2244889.16     13371221.06      2244641.74     13370921.55
      2243717.27     13371030.06
#Sta/Elev= 30
    4280  234.22  4289.9  234.38  4326.2  233.76  4345.7   234.1  4405.3  232.04
  4504.7  228.54    4532  228.38  4560.7  226.62  4582.9  226.68  4589.4  225.84
    4661     224  4692.7  222.66  4732.9  221.89  4752.5  221.78  4757.5  222.24
  4773.2   221.5  4793.4   221.4  4803.4  220.67  4813.5  220.76  4833.6  219.51
  4840.7  218.35  4853.8  218.11  4882.4  216.18  4954.5     214  4984.7  214.39
    4997  213.86  4999.8  213.36    5003  213.86  5246.4  219.32  5599.3  224.95
#Mann= 7 ,-1 , 0
    4280     .05       0  4289.9      .1       0  4345.7     .05       0
  4405.3      .1       0  4882.4     .05       0    4997     .03       0
    5003     .05       0
Bank Sta=4997,5003
XS Rating Curve= 0 ,0
Exp/Cntr=0.3,0.1

Type RM Length L Ch R = 1 ,29233   ,494,494,494
BEGIN DESCRIPTION:
ROCK QUARRY BRANCH 52.0
END DESCRIPTION:
XS GIS Cut Line= 3
      2244889.16     13371221.06      2244641.74     13370921.55
      2243717.27     13371030.06
#Sta/Elev= 30
    4280  234.22  4289.9  234.38  4326.2  233.76  4345.7   234.1  4405.3  232.04
  4504.7  228.54    4532  228.38  4560.7  226.62  4582.9  226.68  4589.4  225.84
    4661     224  4692.7  222.66  4732.9  221.89  4752.5  221.78  4757.5  222.24
  4793.4   221.4  4803.4  220.67  4813.5  220.76  4833.6  219.51  4840.7  218.35
  4853.8  218.11  4882.4  216.18  4954.5     214  4984.7  214.39  5001.8  213.86
  5004.5  213.36  5007.8  213.86    5035   214.7  5246.4  219.32  5599.3  224.95
#Mann= 7 ,-1 , 0
    4280     .05       0  4289.9      .1       0  4345.7     .05       0
  4405.3      .1       0  4882.4     .05       0  5001.8     .03       0
  5007.8     .05       0
Bank Sta=4984.7,5035
XS Rating Curve= 0 ,0
Exp/Cntr=0.3,0.1

Type RM Length L Ch R = 1 ,28755   ,537,537,537
BEGIN DESCRIPTION:
ROCK QUARRY BRANCH 51.0
END DESCRIPTION:
XS GIS Cut Line= 3
      2245006.35     13370439.78      2244468.13     13370413.74
       2243531.7     13370704.21
#Sta/Elev= 30
  4240.7  220.53  4299.4  219.27  4329.4   219.2  4369.5  217.74  4379.5  216.95
  4409.6  216.59  4439.6  215.45  4539.7  214.73  4549.7  213.53  4559.7   213.4
  4569.7   214.6  4619.8   214.1  4657.7  214.56  4731.7   214.4  4832.3  214.59
  4916.1   213.8  4925.8   213.3    4997  211.32  4999.8  210.82    5003  211.32
  5077.7  212.58  5104.6  213.56  5115.5  213.39  5167.4  215.15  5222.8  215.78
  5397.7  218.34  5523.4  220.72  5575.7  221.19  5647.3   223.1    5760  225.18
#Mann= 7 ,-1 , 0
  4240.7     .05       0  4657.7      .1       0  4731.7     .05       0
  4925.8     .07       0    4997     .07       0    5003     .07       0
  5222.8     .05       0
Bank Sta=4997,5003
XS Rating Curve= 0 ,0
Exp/Cntr=0.3,0.1

Type RM Length L Ch R = 1 ,28739   ,537,537,537
BEGIN DESCRIPTION:
ROCK QUARRY BRANCH 51.0
END DESCRIPTION:
XS GIS Cut Line= 3
      2245006.35     13370439.78      2244468.13     13370413.74
       2243531.7     13370704.21
#Sta/Elev= 30
  4240.7  220.53  4299.4  219.27  4329.4   219.2  4379.5  216.95  4409.6  216.59
  4439.6  215.45  4539.7  214.73  4549.7  213.53  4559.7   213.4  4569.7   214.6
  4619.8   214.1  4657.7  214.56  4731.7   214.4  4832.3  214.59  4916.1   213.8
  4925.8   213.3  4968.4  211.91  4989.4  211.81  4996.9  211.32  4999.6  210.82
  5002.9  211.32  5020.8   211.8  5077.7  212.58  5104.6  213.56  5115.5  213.39
  5167.4  215.15  5222.8  215.78  5575.7  221.19  5647.3   223.1    5760  225.18
#Mann= 7 ,-1 , 0
  4240.7     .05       0  4657.7      .1       0  4731.7     .05       0
  4925.8     .07       0  4996.9     .07       0  5002.9     .07       0
  5222.8     .05       0
Bank Sta=4989.4,5020.8
XS Rating Curve= 0 ,0
Exp/Cntr=0.3,0.1

Type RM Length L Ch R = 1 ,28218   ,170,170,170
BEGIN DESCRIPTION:
ROCK QUARRY BRANCH 50.0
END DESCRIPTION:
XS GIS Cut Line= 5
      2245136.58     13370066.53      2244754.59     13369988.39
      2244567.95     13369971.03      2244133.93     13370109.92
      2243482.87     13370509.23
#Sta/Elev= 30
  4260.6  231.69  4300.3     232  4380.3   228.1  4481.2  226.82  4494.2  225.03
  4531.7  223.46  4545.2  224.26  4582.1  222.42  4626.9  222.51  4632.6  219.71
  4637.7  219.21  4683.5  219.97  4697.6  218.89  4707.6  216.05  4731.7  214.94
  4780.7  212.43  4857.9  208.91  4975.9  209.12  4985.6  208.03    4997  207.92
  4999.8  207.42    5003  207.92  5027.2   209.6    5154  212.77  5298.6  216.91
  5388.7  218.07    5416  218.13  5568.7  219.55  5775.8   220.5  6057.4  225.24
#Mann= 13 ,-1 , 0
  4260.6     .05       0  4683.5      .1       0  4731.7     .05       0
  4780.7      .1       0  4857.9     .05       0  4985.6     .12       0
    4997     .07       0    5003     .12       0    5154     .05       0
  5298.6     .12       0  5388.7     .05       0    5416     .12       0
  5568.7     .05       0
Bank Sta=4997,5003
XS Rating Curve= 0 ,0
Exp/Cntr=0.3,0.1

Type RM Length L Ch R = 1 ,28202   ,170,170,170
BEGIN DESCRIPTION:
ROCK QUARRY BRANCH 50.0
END DESCRIPTION:
XS GIS Cut Line= 5
      2245136.58     13370066.53      2244754.59     13369988.39
      2244567.95     13369971.03      2244133.93     13370109.92
      2243482.87     13370509.23
#Sta/Elev= 30
  4260.6  231.69  4300.3     232  4380.3   228.1  4481.2  226.82  4531.7  223.46
  4545.2  224.26  4582.1  222.42  4626.9  222.51  4632.6  219.71  4637.7  219.21
  4683.5  219.97  4697.6  218.89  4707.6  216.05  4731.7  214.94  4780.7  212.43
  4857.9  208.91  4975.9  209.12  4985.6  208.02  4992.7  207.92  4995.4  207.42
  4998.7  207.92  5002.8  209.12  5104.5  210.51    5154  212.77  5298.6  216.91
  5388.7  218.07    5416  218.13  5568.7  219.55  5775.8   220.5  6057.4  225.24
#Mann= 13 ,-1 , 0
  4260.6     .05       0  4683.5      .1       0  4731.7     .05       0
  4780.7      .1       0  4857.9     .05       0  4985.6     .12       0
  4992.7     .07       0  4998.7     .12       0    5154     .05       0
  5298.6     .12       0  5388.7     .05       0    5416     .12       0
  5568.7     .05       0
Bank Sta=4975.9,5002.8
XS Rating Curve= 0 ,0
Exp/Cntr=0.3,0.1

Type RM Length L Ch R = 1 ,28048   ,170,170,170
BEGIN DESCRIPTION:
Mapping XS ce08cd12
END DESCRIPTION:
XS GIS Cut Line= 5
      2245048.12     13369948.87      2244622.77     13369870.74
      2244388.39     13369862.06      2244093.25      13369931.5
      2243439.51     13370283.52
#Sta/Elev= 30
  4421.4  230.73  4645.5   222.7  4686.4   216.8  4739.5  218.05  4747.2  220.72
  4757.3  218.72  4848.5   217.9  4858.9  220.55    4929     216    4939  212.41
  4989.3  207.54    4997  207.46  4999.8  206.96    5003  207.46    5039  209.82
  5069.1  219.84  5109.6  221.48  5128.1  219.25  5140.5  221.37  5181.6   222.4
    5218  220.83  5223.1  222.51  5260.4  218.95  5265.5  222.28  5302.8  218.66
  5345.1   222.2  5387.7   218.4    5518  221.13  5901.8   223.9  6134.1     228
#Mann= 7 ,-1 , 0
  4421.4     .05       0  4848.5      .1       0  4989.3     .12       0
    4997     .07       0    5003     .12       0  5387.7     .05       0
  5901.8      .1       0
Bank Sta=4997,5003
XS Rating Curve= 0 ,0
Exp/Cntr=0.3,0.1

Type RM Length L Ch R = 1 ,28032   ,170,170,170
BEGIN DESCRIPTION:
Mapping XS ce08cd12
END DESCRIPTION:
XS GIS Cut Line= 5
      2245048.12     13369948.87      2244622.77     13369870.74
      2244388.39     13369862.06      2244093.25      13369931.5
      2243439.51     13370283.52
#Sta/Elev= 30
  4421.4  230.73  4645.5   222.7  4686.4   216.8  4739.5  218.05  4747.2  220.72
  4757.3  218.72  4848.5   217.9  4858.9  220.55    4929     216    4939  212.41
    4959  210.03  4989.3  207.54    4996  207.46  4998.8  206.96    5002  207.46
  5002.4  207.49    5039  209.82  5069.1  219.84  5109.6  221.48  5128.1  219.25
  5140.5  221.37    5218  220.83  5223.1  222.51  5260.4  218.95  5265.5  222.28
  5302.8  218.66  5345.1   222.2  5387.7   218.4  5901.8   223.9  6134.1     228
#Mann= 8 ,-1 , 0
  4421.4     .05       0  4848.5      .1       0  4989.3     .12       0
    4996     .07       0    5002     .12       0  5002.4      .1       0
  5387.7     .05       0  5901.8      .1       0
Bank Sta=4959,5039
XS Rating Curve= 0 ,0
Exp/Cntr=0.3,0.1

Type RM Length L Ch R = 1 ,27878   ,318,318,318
BEGIN DESCRIPTION:
ROCK QUARRY BRANCH 49.0
END DESCRIPTION:
XS GIS Cut Line= 3
      2244987.69     13369896.84      2244487.72     13369696.85
      2243687.73     13369596.86
#Sta/Elev= 30
  4461.6  228.27  4476.9  227.71  4500.6  226.68    4506  227.69  4524.8   225.6
  4534.4  225.34  4590.8  224.04  4601.6  225.24  4623.1  223.36  4632.5  221.53
  4637.9  222.23  4655.4  217.18  4662.2  216.16  4845.2  210.92  4936.8  209.95
  4990.7  208.11    4997  207.05  4999.8  206.55    5003  207.05  5010.2  208.15
  5030.3  207.05  5050.5  209.13  5060.5  208.38  5118.5  210.51  5151.2   210.6
    5252  215.32  5379.1  218.54  5483.8  221.85  5774.3  227.52  5806.3  227.99
#Mann= 8 ,-1 , 0
  4461.6     .05       0  4476.9      .1       0  4534.4     .05       0
  4845.2      .1       0    4997     .07       0    5003      .1       0
  5379.1     .05       0  5774.3      .1       0
Bank Sta=4997,5003
XS Rating Curve= 0 ,0
Exp/Cntr=0.3,0.1

Type RM Length L Ch R = 1 ,27862   ,319,319,319
BEGIN DESCRIPTION:
ROCK QUARRY BRANCH 49.0
END DESCRIPTION:
XS GIS Cut Line= 3
      2244987.69     13369896.84      2244487.72     13369696.85
      2243687.73     13369596.86
#Sta/Elev= 30
  4461.6  228.27  4476.9  227.71  4500.6  226.68    4506  227.69  4524.8   225.6
  4534.4  225.34  4590.8  224.04  4601.6  225.24  4623.1  223.36  4632.5  221.53
  4637.9  222.23  4655.4  217.18  4662.2  216.16  4845.2  210.92  4907.2  210.68
  4955.7  209.34  4997.4  207.25  5010.2  208.15  5027.3  207.05  5030.1  206.55
  5033.3  207.05  5050.5  209.13  5060.5  208.38  5118.5  210.51  5151.2   210.6
    5252  215.32  5379.1  218.54  5483.8  221.85  5774.3  227.52  5806.3  227.99
#Mann= 8 ,-1 , 0
  4461.6     .05       0  4476.9      .1       0  4534.4     .05       0
  4845.2      .1       0  5027.3     .07       0  5033.3      .1       0
  5379.1     .05       0  5774.3      .1       0
Bank Sta=4955.7,5050.5
XS Rating Curve= 0 ,0
Exp/Cntr=0.3,0.1

Type RM Length L Ch R = 1 ,27560   ,452,452,452
BEGIN DESCRIPTION:
ROCK QUARRY BRANCH 48.0
END DESCRIPTION:
XS GIS Cut Line= 3
      2245255.35     13369631.21      2244888.89     13369399.54
      2243722.36     13369382.69
#Sta/Elev= 30
  4189.9  230.07    4212  230.04  4329.1  226.21  4409.6  224.59  4553.9  218.94
  4654.6  216.76  4664.6  215.28  4774.6  214.24  4814.6  212.33  4884.6  211.27
  4894.6  210.04  4924.7  209.92  4984.7  207.63    4997  205.32  4999.8  204.82
    5003  205.32  5004.7   206.2  5024.7  206.99  5104.7  207.54  5224.7  213.31
  5274.7  214.56  5314.7   216.6  5344.7   216.4  5354.7  217.66  5424.7  219.94
  5474.7  220.46  5744.7  226.63  5764.7  226.08  5784.7  227.66  5790.1  226.83
#Mann= 3 ,-1 , 0
  4189.9      .1       0    4997     .07       0    5003      .1       0
Bank Sta=4997,5003
XS Rating Curve= 0 ,0
Exp/Cntr=0.3,0.1

Type RM Length L Ch R = 1 ,27543   ,452,452,452
BEGIN DESCRIPTION:
ROCK QUARRY BRANCH 48.0
END DESCRIPTION:
XS GIS Cut Line= 3
      2245255.35     13369631.21      2244888.89     13369399.54
      2243722.36     13369382.69
#Sta/Elev= 30
  4189.9  230.07    4212  230.04  4306.2  227.59  4329.1  226.21  4409.6  224.59
  4553.9  218.94  4654.6  216.76  4664.6  215.28  4774.6  214.24  4814.6  212.33
  4884.6  211.27  4894.6  210.04  4924.7  209.92  4984.7  207.63  4991.7  205.32
  4994.4  204.82  4997.7  205.32  5024.7  206.99  5104.7  207.54  5224.7  213.31
  5274.7  214.56  5314.7   216.6  5344.7   216.4  5354.7  217.66  5424.7  219.94
  5474.7  220.46  5744.7  226.63  5764.7  226.08  5784.7  227.66  5790.1  226.83
#Mann= 3 ,-1 , 0
  4189.9      .1       0  4991.7     .07       0  4997.7      .1       0
Bank Sta=4984.7,5024.7
XS Rating Curve= 0 ,0
Exp/Cntr=0.3,0.1

Type RM Length L Ch R = 1 ,27108   ,366,366,366
BEGIN DESCRIPTION:
ROCK QUARRY BRANCH 47.0
END DESCRIPTION:
XS GIS Cut Line= 2
      2245533.35     13368999.37       2243747.3     13368986.73
#Sta/Elev= 30
  4091.7  221.21  4197.3  218.28  4277.3  214.87  4317.3   214.8  4427.3  212.62
  4457.3  210.22  4477.3  211.42  4527.3  209.43  4612.7  208.68  4650.7  208.07
  4757.3  206.63  4767.3  207.13  4857.4  205.17  4899.7  205.36    4929   205.3
  4957.4  205.62  4987.4   204.6    4997  203.39  4999.8  202.89    5003  203.39
  5027.4  205.09  5117.4  208.71  5137.4  208.62  5167.4  210.62  5267.4  212.11
  5327.4  215.37  5377.4  215.52  5417.4  217.17  5587.4   220.4  5877.8  224.32
#Mann= 7 ,-1 , 0
  4091.7      .1       0  4612.7     .16       0  4650.7      .1       0
  4899.7     .16       0    4929      .1       0    4997     .07       0
    5003      .1       0
Bank Sta=4997,5003
XS Rating Curve= 0 ,0
Exp/Cntr=0.3,0.1

Type RM Length L Ch R = 1 ,27091   ,365,365,365
BEGIN DESCRIPTION:
ROCK QUARRY BRANCH 47.0
END DESCRIPTION:
XS GIS Cut Line= 2
      2245533.35     13368999.37       2243747.3     13368986.73
#Sta/Elev= 30
  4091.7  221.21  4197.3  218.28  4277.3  214.87  4317.3   214.8  4427.3  212.62
  4457.3  210.22  4477.3  211.42  4527.3  209.43  4612.7  208.68  4650.7  208.07
  4757.3  206.63  4767.3  207.13  4857.4  205.17  4899.7  205.36    4929   205.3
  4957.4  205.62  5004.4  203.39  5007.1  202.89  5010.4  203.39  5027.4  205.09
  5047.4   205.9  5117.4  208.71  5137.4  208.62  5167.4  210.62  5267.4  212.11
  5327.4  215.37  5377.4  215.52  5417.4  217.17  5587.4   220.4  5877.8  224.32
#Mann= 7 ,-1 , 0
  4091.7      .1       0  4612.7     .16       0  4650.7      .1       0
  4899.7     .16       0    4929      .1       0  5004.4     .07       0
  5010.4      .1       0
Bank Sta=4957.4,5047.4
XS Rating Curve= 0 ,0
Exp/Cntr=0.3,0.1

Type RM Length L Ch R = 1 ,26742   ,548,548,548
BEGIN DESCRIPTION:
ROCK QUARRY BRANCH 46.0
END DESCRIPTION:
XS GIS Cut Line= 2
      2245634.43     13368780.33      2243871.07     13368750.87
#Sta/Elev= 30
  4242.4  219.46  4309.1  216.14  4459.1  212.74  4489.1  212.55  4559.2  211.11
  4569.2  211.57  4579.2  211.29  4589.2  210.37  4629.2  209.19  4823.1   204.3
  4879.2  202.96  4921.3  202.74  4959.2     203  4969.2  202.08  4989.2  201.08
    4997  201.08  4999.8  200.58    5003  201.08  5009.2  202.79  5019.2  202.51
  5095.5  204.17  5159.2  206.04  5329.3  209.43  5346.2  210.28  5409.3  211.47
  5639.3  215.27  5689.3  215.62  5849.3   218.2  5919.3  218.84    6006  220.49
#Mann= 6 ,-1 , 0
  4242.4      .1       0  4823.1     .16       0  4921.3      .1       0
    4997     .07       0    5003      .1       0  5095.5     .05       0
Bank Sta=4997,5003
XS Rating Curve= 0 ,0
Exp/Cntr=0.3,0.1

Type RM Length L Ch R = 1 ,26726   ,548,548,548
BEGIN DESCRIPTION:
ROCK QUARRY BRANCH 46.0
END DESCRIPTION:
XS GIS Cut Line= 2
      2245634.43     13368780.33      2243871.07     13368750.87
#Sta/Elev= 30
  4242.4  219.46  4309.1  216.14  4429.1  213.68  4459.1  212.74  4489.1  212.55
  4559.2  211.11  4569.2  211.57  4579.2  211.29  4589.2  210.37  4629.2  209.19
  4823.1   204.3  4879.2  202.96  4921.3  202.74  4959.2     203  4986.2  201.08
    4989  200.58  4992.2  201.08  4999.2  202.29  5009.2  202.79  5019.2  202.51
  5095.5  204.17  5159.2  206.04  5329.3  209.43  5346.2  210.28  5409.3  211.47
  5639.3  215.27  5689.3  215.62  5849.3   218.2  5919.3  218.84    6006  220.49
#Mann= 6 ,-1 , 0
  4242.4      .1       0  4823.1     .16       0  4921.3      .1       0
  4986.2     .07       0  4992.2      .1       0  5095.5     .05       0
Bank Sta=4959.2,5009.2
XS Rating Curve= 0 ,0
Exp/Cntr=0.3,0.1

Type RM Length L Ch R = 1 ,26194   ,443,443,443
BEGIN DESCRIPTION:
ROCK QUARRY BRANCH 45.0
END DESCRIPTION:
XS GIS Cut Line= 2
      2245727.11     13368531.79      2244467.64     13368127.41
#Sta/Elev= 30
  4433.5  218.85  4579.9   215.8  4660.5   211.7  4705.9   211.7  4737.4  209.73
  4747.9  210.47  4779.5  208.46  4788.9  208.91    4811  206.05  4890.5  200.62
    4937  199.52    4979  199.87  4992.1  199.37    4997  198.02  4999.8  197.52
    5003  198.02  5018.9  200.27  5078.8  200.75  5180.6  202.09  5254.2  201.54
  5304.6  204.35  5325.6  207.19  5336.1  210.15  5350.5  212.34  5357.1  215.38
  5377.4  218.15  5399.1  219.13    5479   216.3  5516.3  216.08  5756.3  222.28
#Mann= 5 ,-1 , 0
  4433.5      .1       0    4997     .07       0    5003      .1       0
  5078.8     .05       0  5180.6      .1       0
Bank Sta=4997,5003
XS Rating Curve= 0 ,0
Exp/Cntr=0.3,0.1

Type RM Length L Ch R = 1 ,26178   ,443,443,443
BEGIN DESCRIPTION:
ROCK QUARRY BRANCH 45.0
END DESCRIPTION:
XS GIS Cut Line= 2
      2245727.11     13368531.79      2244467.64     13368127.41
#Sta/Elev= 30
  4433.5  218.85  4579.9   215.8  4660.5   211.7  4705.9   211.7  4737.4  209.73
  4747.9  210.47  4779.5  208.46  4788.9  208.91    4811  206.05  4890.5  200.62
    4937  199.52    4979  199.87  4992.1  199.37    4997  198.02  4999.8  197.52
    5003  198.02  5018.9  200.27  5078.8  200.75  5180.6  202.09  5254.2  201.54
  5304.6  204.35  5325.6  207.19  5336.1  210.15  5350.5  212.34  5357.1  215.38
  5377.4  218.15  5399.1  219.13    5479   216.3  5516.3  216.08  5756.3  222.28
#Mann= 5 ,-1 , 0
  4433.5      .1       0    4997     .07       0    5003      .1       0
  5078.8     .05       0  5180.6      .1       0
Bank Sta=4979,5018.9
XS Rating Curve= 0 ,0
Exp/Cntr=0.3,0.1

Type RM Length L Ch R = 1 ,25751   ,414,414,414
BEGIN DESCRIPTION:
ROCK QUARRY BRANCH 44.0
END DESCRIPTION:
XS GIS Cut Line= 3
      2245638.64     13367992.61      2245423.86     13367958.92
      2244535.05     13368013.68
#Sta/Elev= 30
  4431.3  214.89  4436.7  214.98  4442.4   213.9  4482.8  212.86  4499.4  211.09
  4567.1  209.53  4594.2  207.57  4612.5  207.49  4761.8  203.33  4859.7  201.71
  4885.3  200.82  4925.4  198.02  4975.5  198.35    4997   196.5  4999.8     196
    5003   196.5  5035.6  198.31  5085.7  198.83  5105.7  198.28  5125.7  202.01
  5155.8  205.01  5165.8  207.26  5175.8  208.29  5182.6  210.37  5187.6  209.75
  5225.9  213.22  5356.2  214.24  5446.4  217.07  5496.5  219.74  5539.2  220.96
#Mann= 5 ,-1 , 0
  4431.3      .1       0  4612.5     .05       0  4761.8      .1       0
    4997     .07       0    5003      .1       0
Bank Sta=4997,5003
XS Rating Curve= 0 ,0
Exp/Cntr=0.3,0.1

Type RM Length L Ch R = 1 ,25735   ,415,415,415
BEGIN DESCRIPTION:
ROCK QUARRY BRANCH 44.0
END DESCRIPTION:
XS GIS Cut Line= 3
      2245638.64     13367992.61      2245423.86     13367958.92
      2244535.05     13368013.68
#Sta/Elev= 30
  4431.3  214.89  4436.7  214.98  4442.4   213.9  4482.8  212.86  4499.4  211.09
  4567.1  209.53  4594.2  207.57  4612.5  207.49  4761.8  203.33  4859.7  201.71
  4885.3  200.82  4925.4  198.02  4975.5  198.35  4992.5   196.5  4995.3     196
  4998.5   196.5  5035.6  198.31  5085.7  198.83  5105.7  198.28  5125.7  202.01
  5155.8  205.01  5165.8  207.26  5175.8  208.29  5182.6  210.37  5187.6  209.75
  5225.9  213.22  5356.2  214.24  5446.4  217.07  5496.5  219.74  5539.2  220.96
#Mann= 5 ,-1 , 0
  4431.3      .1       0  4612.5     .05       0  4761.8      .1       0
  4992.5     .07       0  4998.5      .1       0
Bank Sta=4975.5,5035.6
XS Rating Curve= 0 ,0
Exp/Cntr=0.3,0.1

Type RM Length L Ch R = 1 ,25337   ,557,557,557
BEGIN DESCRIPTION:
ROCK QUARRY BRANCH 43.0
END DESCRIPTION:
XS GIS Cut Line= 3
      2245613.42     13367744.09      2245457.55     13367664.06
      2244543.48     13367516.62
#Sta/Elev= 30
  4474.2  214.29    4477  215.86  4482.7  214.08  4491.8  215.51  4504.8   214.8
  4521.4  216.25    4527  214.23  4559.3  218.86    4588  217.56  4610.2  213.96
  4615.8  211.53  4632.3  208.58  4658.8  206.39  4669.5  203.64  4701.4   201.7
  4829.9  199.13  4932.9  197.33    4997  194.74  4999.8  194.24    5003  194.74
  5013.9  196.31  5106.5  196.42  5291.8  204.53  5307.6  206.18  5358.7  207.43
  5408.9     210  5415.4  211.41  5449.5  212.46  5500.1   217.3  5575.3  221.03
#Mann= 5 ,-1 , 0
  4474.2      .1       0  4701.4     .05       0  4829.9      .1       0
    4997     .07       0    5003      .1       0
Bank Sta=4997,5003
XS Rating Curve= 0 ,0
Exp/Cntr=0.3,0.1

Type RM Length L Ch R = 1 ,25320   ,556,556,556
BEGIN DESCRIPTION:
ROCK QUARRY BRANCH 43.0
END DESCRIPTION:
XS GIS Cut Line= 3
      2245613.42     13367744.09      2245457.55     13367664.06
      2244543.48     13367516.62
#Sta/Elev= 30
  4474.2  214.29    4477  215.86  4482.7  214.08  4491.8  215.51  4504.8   214.8
  4521.4  216.25    4527  214.23  4559.3  218.86    4588  217.56  4610.2  213.96
  4615.8  211.53  4632.3  208.58  4658.8  206.39  4669.5  203.64  4701.4   201.7
  4829.9  199.13  4963.2  196.34  4990.6  194.74  4993.4  194.24  4996.6  194.74
  5013.9  196.31  5101.4  196.25  5277.3  203.84  5307.6  206.18  5408.9     210
  5415.4  211.41  5420.5  210.77  5449.5  212.46  5500.1   217.3  5575.3  221.03
#Mann= 5 ,-1 , 0
  4474.2      .1       0  4701.4     .05       0  4829.9      .1       0
  4990.6     .07       0  4996.6      .1       0
Bank Sta=4963.2,5013.9
XS Rating Curve= 0 ,0
Exp/Cntr=0.3,0.1

Type RM Length L Ch R = 1 ,24780   ,362,362,362
BEGIN DESCRIPTION:
ROCK QUARRY BRANCH 42.0
END DESCRIPTION:
XS GIS Cut Line= 4
      2245687.74     13367296.86      2244886.37     13367020.04
      2244735.33     13366967.96      2244506.17      13367061.7
#Sta/Elev= 30
  4347.3  217.07  4362.9   217.6  4368.5  216.23  4425.3  211.91  4442.5   209.6
  4544.7  202.82  4622.4   201.3  4726.5  197.02  4856.6  194.26  4913.6  194.94
  4944.8  193.29  4970.7  194.35    4997  193.29  4999.8  192.79    5003  193.29
  5163.1  202.03  5251.4  211.74  5257.2  213.49  5282.6  216.06  5308.5  216.97
  5313.8   218.3  5390.9  217.07  5396.3  218.37  5414.9  218.12  5449.7  220.04
  5497.7  220.78  5521.7  219.37  5551.1  220.55  5568.4  219.66  5602.5  220.43
#Mann= 3 ,-1 , 0
  4347.3      .1       0    4997     .07       0    5003      .1       0
Bank Sta=4997,5003
XS Rating Curve= 0 ,0
Exp/Cntr=0.3,0.1

Type RM Length L Ch R = 1 ,24764   ,362,362,362
BEGIN DESCRIPTION:
ROCK QUARRY BRANCH 42.0
END DESCRIPTION:
XS GIS Cut Line= 4
      2245687.74     13367296.86      2244886.37     13367020.04
      2244735.33     13366967.96      2244506.17      13367061.7
#Sta/Elev= 30
  4347.3  217.07  4362.9   217.6  4368.5  216.23  4442.5   209.6  4544.7  202.82
  4622.4   201.3  4726.5  197.02  4865.7  194.12  4913.6  194.94  4941.8  193.29
  4944.6  192.79  4947.8  193.29  4982.1  194.31  5007.2  193.66  5033.1   195.1
  5163.1  202.03  5251.4  211.74  5257.2  213.49  5282.6  216.06  5308.5  216.97
  5313.8   218.3  5390.9  217.07  5396.3  218.37  5414.9  218.12  5449.7  220.04
  5497.7  220.78  5521.7  219.37  5551.1  220.55  5568.4  219.66  5602.5  220.43
#Mann= 3 ,-1 , 0
  4347.3      .1       0  4941.8     .07       0  4947.8      .1       0
Bank Sta=4982.1,5033.1
XS Rating Curve= 0 ,0
Exp/Cntr=0.3,0.1

Type RM Length L Ch R = 1 ,24418   ,484,484,484
BEGIN DESCRIPTION:
ROCK QUARRY BRANCH 41.0
END DESCRIPTION:
XS GIS Cut Line= 4
      2245875.92     13367040.86       2245344.7     13366801.29
      2244891.58     13366686.71      2244516.57     13366723.17
#Sta/Elev= 30
  4259.1  219.28    4287  218.77  4300.4  218.46  4322.9  216.17  4334.5   216.4
  4366.8  214.25  4432.6  212.22  4496.5  208.68  4501.9  209.21  4509.4   207.9
  4525.1   207.9  4564.3  205.12  4761.7  196.36  4890.3  192.64  4959.6  193.29
    4997  191.66  4999.8  191.16    5003  191.66  5005.8  192.58  5014.1     193
  5089.4   195.3  5169.9  198.01  5217.9  200.64  5302.9  203.08  5308.6  203.94
  5353.3  205.72  5462.3  208.96    5514  209.25  5671.1  215.24    5686  214.94
#Mann= 6 ,-1 , 0
  4259.1     .05       0    4287      .1       0    4997     .07       0
    5003      .1       0  5089.4     .05       0  5217.9      .1       0
Bank Sta=4997,5003
XS Rating Curve= 0 ,0
Exp/Cntr=0.3,0.1

Type RM Length L Ch R = 1 ,24402   ,484,484,484
BEGIN DESCRIPTION:
ROCK QUARRY BRANCH 41.0
END DESCRIPTION:
XS GIS Cut Line= 4
      2245875.92     13367040.86       2245344.7     13366801.29
      2244891.58     13366686.71      2244516.57     13366723.17
#Sta/Elev= 30
  4259.1  219.28    4287  218.77  4300.4  218.46  4322.9  216.17  4334.5   216.4
  4366.8  214.25  4432.6  212.22  4496.5  208.68  4501.9  209.21  4509.4   207.9
  4525.1   207.9  4564.3  205.12  4761.7  196.36  4890.3  192.64  4959.6  193.29
  4990.4  191.66  4993.2  191.16  4996.4  191.66  5024.4  193.16  5089.4   195.3
  5169.9  198.01  5217.9  200.64  5302.9  203.08  5308.6  203.94  5353.3  205.72
  5462.3  208.96    5514  209.25  5534.1  210.55  5671.1  215.24    5686  214.94
#Mann= 6 ,-1 , 0
  4259.1     .05       0    4287      .1       0  4990.4     .07       0
  4996.4      .1       0  5089.4     .05       0  5217.9      .1       0
Bank Sta=4959.6,5024.4
XS Rating Curve= 0 ,0
Exp/Cntr=0.3,0.1
