HEC-RAS study SULPHUR CREEK.prj: SULPHUR CREEK Base Level Engineering

--- SULPHUR CREEK.g01 (geometry) --- (continued)

Type RM Length L Ch R = 1 ,159497  ,400,400,400
BEGIN DESCRIPTION:
SULPHUR CREEK 179.0
END DESCRIPTION:
XS GIS Cut Line= 4
      2295465.84      13436018.4      2294735.35     13436594.12
      2294202.97     13437027.46      2294215.35     13437857.02
#Sta/Elev= 30
  3788.9  373.88  4085.5  369.09  4377.3  362.11  4406.2   360.5    4427  360.99
  4455.9  359.12    4605  358.76  4797.2     354  4811.5  354.89  4840.9  354.72
  4875.5  354.07  4968.1  354.76  4988.9  353.51  5000.3  347.31    5003  346.81
  5006.3  347.31  5017.7  347.57  5025.4  353.61  5038.5     354  5074.9  353.51
  5116.8  355.02  5209.4  353.67  5238.2  357.51  5273.3  359.65  5407.6  361.61
  5444.8   362.6  5454.8  364.01  5494.9  363.19  5874.9  367.68  6235.1  369.49
#Mann= 5 ,-1 , 0
  3788.9     .05       0  4840.9      .1       0  5000.3     .07       0
  5006.3      .1       0  5074.9     .05       0
Bank Sta=4968.1,5038.5
XS Rating Curve= 0 ,0
Exp/Cntr=0.3,0.1

Type RM Length L Ch R = 1 ,159097  ,482,482,482
BEGIN DESCRIPTION:
SULPHUR CREEK 178.0
END DESCRIPTION:
XS GIS Cut Line= 3
      2295240.28     13435929.15      2294242.62     13436536.06
      2292617.36     13436660.76
#Sta/Elev= 30
    4029  368.93    4348  363.06  4654.1  352.85  4787.3  353.17  4801.3  352.33
  4813.2  347.05    4816  346.55  4819.2  347.05  4822.6  352.13    4902  353.41
  4960.2  349.74  4981.5   351.8  5018.3  350.49    5062  353.12  5192.7  350.33
  5274.7  350.89  5304.2  353.12  5351.6  356.35  5405.3  357.35  5422.3  350.62
  5462.4  354.63  5535.8  355.22  5552.7  352.59  5582.8  355.61  5632.9  354.82
  5753.3  359.65  5938.3  359.82  6274.8  360.96  6355.1  359.68  6826.8  369.26
#Mann= 7 ,-1 , 0
    4029     .05       0  4787.3      .1       0  4813.2     .07       0
  4819.2      .1       0  5304.2     .05       0  5351.6      .1       0
  5938.3     .05       0
#XS Ineff= 2 ,-1
 5396.04 5807.64  357.54  6274.4  6461.1  360.97
Permanent Ineff=
       T       T
Bank Sta=4902,5062
XS Rating Curve= 0 ,0
Exp/Cntr=0.3,0.1

Type RM Length L Ch R = 1 ,158615  ,784,784,784
BEGIN DESCRIPTION:
SULPHUR CREEK 177.0
END DESCRIPTION:
XS GIS Cut Line= 4
      2295069.79     13435671.46      2294117.92     13436207.67
      2293619.11     13436307.43      2292525.93     13436502.79
#Sta/Elev= 30
    3956  367.22  4732.1  356.36  4941.2  351.58  4958.9  351.64  4990.8  349.64
  4993.5  346.56  4996.3  346.06  4999.5  346.56  5045.8  351.67    5072   352.1
  5117.9  350.72  5160.9  353.35  5168.9  352.72  5181.3  348.13  5201.7  351.97
  5232.3  352.23  5252.7  349.74  5313.9   354.2  5354.7  354.33    5378  352.89
  5385.3  349.05  5405.6  350.59  5415.8  353.48  5436.2  351.51  5487.2  353.41
  5526.2  358.22  6151.8  359.51  6584.6  369.29  6615.1  372.47  6667.7  371.95
#Mann= 5 ,-1 , 0
    3956     .05       0  4941.2      .1       0  4993.5     .07       0
  4999.5      .1       0  5526.2     .05       0
Bank Sta=4958.9,5072
XS Rating Curve= 0 ,0
Exp/Cntr=0.3,0.1

Type RM Length L Ch R = 1 ,157831  ,570,570,570
BEGIN DESCRIPTION:
SULPHUR CREEK 176.0
END DESCRIPTION:
XS GIS Cut Line= 3
      2295287.77     13435496.86      2294037.72     13435446.85
      2292437.74     13436396.84
#Sta/Elev= 30
  3742.1  382.92  3778.2  374.98  3802.2  372.83  4018.5  368.09  4572.8     360
  4622.9  359.64  4642.9  361.77  4730.7  358.45    4853  354.73  4966.5  348.32
  4968.6  348.11  4983.1  347.81    4998  344.27  5000.7  343.77    5004  344.27
  5016.4  348.41  5074.6  349.56  5139.3  354.36  5373.1  353.49  5591.3  356.53
  5911.9   356.5  6240.1  359.38  6335.6  362.27  6378.5  361.58  6670.8  369.69
  6686.4   372.7  6723.4     371  6760.4  373.95  6824.7  373.65  6853.9  375.98
#Mann= 8 ,-1 , 0
  3742.1      .1       0  3778.2     .05       0  4018.5      .1       0
  4730.7     .05       0  4966.5      .1       0  4968.6     .05       0
    4998     .03       0    5004     .05       0
Bank Sta=4853,5139.3
XS Rating Curve= 0 ,0
Exp/Cntr=0.3,0.1

Type RM Length L Ch R = 1 ,157261  ,547,547,547
BEGIN DESCRIPTION:
SULPHUR CREEK 175.0
END DESCRIPTION:
XS GIS Cut Line= 3
      2295187.68     13434946.86      2293637.72     13435046.85
      2292337.73     13436146.84
#Sta/Elev= 30
  3453.9  379.29  3669.4  372.58  3727.9  370.86  3999.7  364.42  4476.4   357.9
  4772.8  351.82  4856.8  353.03  4896.8  350.93  4936.9  346.27    4977  346.21
  4994.1  341.71  4996.8  341.21  5000.1  341.71  5010.4  342.61  5014.2  345.58
  5042.8  352.73  5063.6  353.56  5127.4  352.16  5177.4  353.93  5264.9  353.64
  5666.8  354.15  6134.8  359.19  6397.4  365.03  6489.7  369.13  6539.7  369.13
  6553.4  371.95  6593.9  370.75  6631.4  373.65  6667.7  373.13    6710   375.2
#Mann= 8 ,-1 , 0
  3453.9      .1       0  3669.4     .05       0  3727.9      .1       0
  3999.7     .05       0  4476.4      .1       0  4994.1     .07       0
  5000.1      .1       0  5264.9     .05       0
Bank Sta=4856.8,5063.6
XS Rating Curve= 0 ,0
Exp/Cntr=0.3,0.1

Type RM Length L Ch R = 1 ,156714  ,517,517,517
BEGIN DESCRIPTION:
SULPHUR CREEK 174.0
END DESCRIPTION:
XS GIS Cut Line= 3
      2294987.68     13433846.87      2293437.72     13434546.85
      2292287.73     13436096.84
#Sta/Elev= 30
  3296.4  376.52  3645.3  368.09    4240  361.93  4440.6  355.55  4884.8  350.55
  4898.3  348.43  4975.1  347.08  4988.3  343.92  4994.3  340.39  5000.2  340.39
  5001.4  338.15  5004.1  337.65  5007.4  338.15  5010.6   342.8  5025.2   345.2
  5119.2  350.04  5240.2  353.26  5418.8  352.94  5621.5  351.89  5705.5  353.62
  5782.7  352.75  6212.5  359.26  6304.5  359.01  6398.2  362.01  6441.5  361.25
  6740.3  369.29  6763.3  372.15  6798.8  370.83  6840.5  373.33  6927.1  373.88
#Mann= 7 ,-1 , 0
  3296.4     .05       0  4440.6      .1       0  4884.8     .07       0
  5119.2      .1       0  5418.8     .05       0  5621.5      .1       0
  5782.7     .05       0
Bank Sta=4884.8,5119.2
XS Rating Curve= 0 ,0
Exp/Cntr=0.3,0.1

Type RM Length L Ch R = 1 ,156197  ,549,549,549
BEGIN DESCRIPTION:
SULPHUR CREEK 173.0
END DESCRIPTION:
XS GIS Cut Line= 3
      2294437.73     13433996.85      2293187.72     13434096.85
      2291887.75     13434896.84
#Sta/Elev= 30
    3766  365.39  4026.8  362.73    4346  355.49  4448.2  352.54  4488.3  345.83
  4528.4  346.39  4568.6  354.31  4598.7  348.21  4638.8  347.39  4839.4  349.97
  4869.5  349.22  4979.9  344.39  4999.7  336.93  5017.5  344.81    5049  346.58
  5078.7  349.11  5113.9  351.24  5348.4   350.5  5375.6  344.04  5506.9  347.43
  5513.2  349.65  5549.5  345.35  5622.9  347.69  5644.1  350.79  5696.3  348.59
  5738.8  351.99  5899.5  353.53  6233.4  359.21  6498.4  368.07  6546.4   368.8
#Mann= 6 ,-1 , 0
    3766     .05       0    4346      .1       0  4839.4     .05       0
    5049      .1       0  5899.5     .05       0  6498.4      .1       0
#XS Ineff= 2 ,-1
    3766 4569.89355.5865 5178.22 5920.79  351.25
Permanent Ineff=
       T       T
Bank Sta=4869.5,5078.7
XS Rating Curve= 0 ,0
Exp/Cntr=0.3,0.1

Type RM Length L Ch R = 1 ,155648  ,515,515,515
BEGIN DESCRIPTION:
SULPHUR CREEK 172.0
END DESCRIPTION:
XS GIS Cut Line= 3
      2294587.74     13432446.84      2293037.72     13433596.85
      2291437.71     13434996.87
#Sta/Elev= 30
    3091  376.35  3434.3  364.35  4098.9  357.74  4206.3  357.15  4227.1  354.03
  4262.6   355.7  4291.8   350.5    4321  354.95  4327.3  350.84  4364.4  349.88
  4383.3  352.84  4771.7  351.72  4834.3  347.26  4878.1  343.74  4971.2  344.34
  4984.5  342.82  4996.1  336.93  4998.9  336.43  5002.1  336.93  5017.9  343.01
  5056.6  346.64    5171  348.03  5453.4  348.18    5517  343.83  5754.9  349.42
  5764.9  349.62  6338.9  358.02  6750.6  368.91  6898.9   373.8  7147.1  376.81
#Mann= 10 ,-1 , 0
    3091     .05       0  4098.9      .1       0  4364.4     .05       0
  4383.3      .1       0  4996.1     .07       0  5002.1      .1       0
    5171     .05       0  5754.9      .1       0  5764.9     .05       0
  6750.6      .1       0
#XS Ineff= 2 ,-1
 3650.57 4386.36  356.28 5277.23 5942.01  348.38
Permanent Ineff=
       T       T
Bank Sta=4834.3,5171
XS Rating Curve= 0 ,0
Exp/Cntr=0.3,0.1

Type RM Length L Ch R = 1 ,155133  ,515,515,515
BEGIN DESCRIPTION:
SULPHUR CREEK 171.0
END DESCRIPTION:
XS GIS Cut Line= 3
      2294487.73     13431946.85      2292937.72     13433096.85
      2291337.75     13434346.83
#Sta/Elev= 30
  3066.9  377.99  3209.8  374.77  3403.1  367.33  3625.1  362.67  3917.2  358.02
  4170.8  356.97  4438.6  354.93  4610.9   353.9  4878.9  348.61  4939.6  346.41
  4960.4  345.07  4993.8  336.01  5001.2  335.81  5003.9  335.31  5007.2  335.81
    5025  339.67  5132.7   344.3  5232.1  346.56  5445.5   348.4  5657.1  346.98
  5708.7  346.34  5781.1  342.42  5874.6   344.7  6243.2  353.07  6485.6  356.29
  6621.3  361.19  6692.7   361.2  6777.7  364.84  6806.7  364.32  7027.3  370.56
#Mann= 9 ,-1 , 0
  3066.9     .05       0  4170.8      .1       0  4438.6     .05       0
  4878.9      .1       0  5001.2     .07       0  5007.2      .1       0
  5132.7     .05       0  5657.1      .1       0  5874.6     .05       0
#XS Ineff= 1 ,-1
 5468.18 6104.67  348.22
Permanent Ineff=
       T
Bank Sta=4939.6,5232.1
XS Rating Curve= 0 ,0
Exp/Cntr=0.3,0.1

Type RM Length L Ch R = 1 ,154618  ,596,596,596
BEGIN DESCRIPTION:
SULPHUR CREEK 170.0
END DESCRIPTION:
XS GIS Cut Line= 3
      2293987.73     13431746.85      2292587.72     13432746.85
      2290987.75     13434296.83
#Sta/Elev= 30
  3280.7  373.13  3510.5  367.63  3632.2  362.35  3844.5  358.66    4018  355.07
  4319.6  353.96  4813.3  347.46  4878.3  345.11  4987.7  340.29  4990.8  333.35
  4993.5  332.85  4996.8  333.35  5004.7  333.44  5008.2  337.44  5015.2  339.35
    5043  342.07  5107.3  341.25    5178  345.15  5658.8  347.04  5810.3     345
  5973.6  341.98  6061.9  348.17  6196.4  354.23  6783.3  361.86  6868.1  365.91
  6896.4  364.52  6967.1  367.84  7002.6  367.25  7108.6  371.59  7228.8  373.49
#Mann= 9 ,-1 , 0
  3280.7     .05       0  3844.5      .1       0  4319.6     .05       0
  4813.3      .1       0  4990.8     .07       0  4996.8      .1       0
    5043     .05       0  5810.3      .1       0  5973.6     .05       0
#XS Ineff= 1 ,-1
 5659.12 6104.67  346.51
Permanent Ineff=
       T
Bank Sta=4878.3,5178
XS Rating Curve= 0 ,0
Exp/Cntr=0.3,0.1

Type RM Length L Ch R = 1 ,154022  ,526,526,526
BEGIN DESCRIPTION:
SULPHUR CREEK 169.0
END DESCRIPTION:
XS GIS Cut Line= 3
       2293737.7     13431646.86      2292187.72     13432346.85
      2290737.71     13433746.87
#Sta/Elev= 30
  3295.8  367.96  3361.8  367.91  3533.2  361.59  3765.8  355.28  3916.7  353.35
  4454.7  349.14  4545.9  347.75  4753.3   345.1  4777.1  343.85  4930.5  341.41
  4987.7   337.8  4993.8  332.72  5000.6  331.99  5003.3  331.49  5006.6  331.99
  5017.7  339.42  5060.2  343.55  5107.8  344.82  5350.1  344.46  5399.6  338.84
  5730.8  346.46  5913.2  348.13  6113.9  351.24  6177.7  348.51  6361.4  354.58
  6792.8  361.87  6891.8  361.71  6976.7  364.93  6990.9   372.1  7012.1  371.28
#Mann= 11 ,-1 , 0
  3295.8     .05       0  3533.2      .1       0  3916.7     .05       0
  4454.7      .1       0  4545.9     .05       0  4753.3      .1       0
  5000.6     .07       0  5006.6      .1       0  5107.8     .05       0
  5730.8      .1       0  5913.2     .05       0
#XS Ineff= 1 ,-1
 5285.01 5819.66  344.33
Permanent Ineff=
       T
Bank Sta=4777.1,5060.2
XS Rating Curve= 0 ,0
Exp/Cntr=0.3,0.1

Type RM Length L Ch R = 1 ,153496  ,543,543,543
BEGIN DESCRIPTION:
SULPHUR CREEK 168.0
END DESCRIPTION:
XS GIS Cut Line= 3
      2293487.74     13431646.85      2291960.78     13431879.37
       2290337.7     13433446.88
#Sta/Elev= 30
  3452.8  361.37  3675.4  355.57  3823.8  353.85  4153.1  350.32  4393.5  348.65
  4412.4   349.7    4841  342.78  4939.8  342.19  4980.2     337  4993.4  330.32
  4996.1  329.82  4999.4  330.32  5004.8  332.04    5012  337.09  5054.4  339.75
  5146.2  340.76  5188.7  336.14  5273.6  341.07  5330.2  342.62  6002.1  345.99
  6369.8  350.52  6501.8  352.46  6525.1  353.08    6886  358.37  6977.9  361.74
  7006.2  360.99  7105.2  364.14  7126.6  366.82  7218.4  367.93  7253.8  370.49
#Mann= 8 ,-1 , 0
  3452.8      .1       0  3823.8     .05       0    4841      .1       0
  4993.4     .07       0  4999.4      .1       0  6369.8     .05       0
  6501.8      .1       0  6525.1     .05       0
Bank Sta=4939.8,5054.4
XS Rating Curve= 0 ,0
Exp/Cntr=0.3,0.1

Type RM Length L Ch R = 1 ,152953  ,567,567,567
BEGIN DESCRIPTION:
SULPHUR CREEK 167.0
END DESCRIPTION:
XS GIS Cut Line= 3
      2293087.73     13430896.85      2291537.72     13431596.85
      2289937.73     13433146.85
#Sta/Elev= 30
  3307.3  359.27    3450  355.72  3587.7  354.27  3591.4  354.29  3731.1  351.97
  4244.1  349.06  4416.9  345.14  4448.4  342.98  4532.5  340.88  4780.2  341.38
  4848.6  339.77  4976.1  337.17  4986.1  336.48  4996.2  329.66    4999  329.16
  5002.2  329.66  5011.5  330.76  5015.1  334.46  5050.4  337.32  5071.7  341.43
    5264     343  5290.3  342.79  5474.8  342.61  5693.4  344.37  6146.7  350.78
  6291.8  350.99  6366.1  351.59  6747.9  357.85  7136.8  369.34  7235.7  373.74
#Mann= 11 ,-1 , 0
  3307.3     .05       0  3587.7      .1       0  3591.4     .05       0
  4848.6      .1       0  4996.2     .07       0  5002.2      .1       0
    5264     .05       0  5290.3      .1       0  5693.4     .05       0
  6291.8      .1       0  6366.1     .05       0
Bank Sta=4780.2,5071.7
XS Rating Curve= 0 ,0
Exp/Cntr=0.3,0.1

Type RM Length L Ch R = 1 ,152386  ,481,481,481
BEGIN DESCRIPTION:
SULPHUR CREEK 166.0
END DESCRIPTION:
XS GIS Cut Line= 3
      2293037.75     13430746.85      2291487.72     13431146.85
       2289887.7     13432696.87
#Sta/Elev= 30
  3383.6   359.7  3718.8  351.66  3792.4  350.84  4292.5  347.91    4592  338.96
  4757.2  340.38  4827.5  338.18  4963.3  334.97  4974.1  335.37  4981.8  329.08
  4985.6  329.08  4988.5  328.24  4991.2  327.74  4994.5  328.24  5005.6  332.55
  5012.6  331.75  5019.8  336.07  5026.7  333.66  5033.9  336.33  5083.3  333.93
  5168.2  334.85  5210.7  336.72    5232  340.02  5282.9  342.21    5395  342.22
  5744.3  342.56    5854  344.42  6021.6   346.6  6738.4  351.83  7212.1  362.44
#Mann= 13 ,-1 , 0
  3383.6     .05       0  3718.8      .1       0  3792.4     .05       0
  4827.5      .1       0  4963.3     .12       0  4985.6      .1       0
  4988.5     .07       0  4994.5      .1       0  5282.9     .05       0
    5395      .1       0  5744.3     .05       0    5854      .1       0
  6021.6     .05       0
Bank Sta=4757.2,5232
XS Rating Curve= 0 ,0
Exp/Cntr=0.3,0.1

Type RM Length L Ch R = 1 ,151905  ,447,447,447
BEGIN DESCRIPTION:
SULPHUR CREEK 165.0
END DESCRIPTION:
XS GIS Cut Line= 3
      2292037.68     13430846.84      2291606.61      13430710.1
      2290487.71     13431696.86
#Sta/Elev= 30
  4558.6  345.63    4632  343.73  4741.3  343.03  4838.1  338.76  4883.8  338.27
  4925.7  335.21  4934.9  335.55  4946.7  332.18  4957.1  336.16  4978.2  337.99
  4988.7  335.08  4996.2  327.11  4998.9  326.61  5002.2  327.11  5004.7  329.17
    5029  330.61  5043.2  335.44  5057.4  335.88  5105.9  336.19  5135.2  337.52
  5156.1  336.84  5163.7  337.87  5206.4  337.65  5270.1  339.52    5596  341.98
  5881.8  340.79  5921.7  340.58  5938.2  339.41  6438.7   345.6  6502.7  347.15
#Mann= 8 ,-1 , 0
  4558.6     .05       0  4957.1     .12       0  4996.2     .07       0
  5002.2     .12       0  5105.9      .1       0  5270.1     .05       0
  5881.8      .1       0  5938.2     .05       0
#XS Ineff= 1 ,-1
  5617.4 6232.67  341.36
Permanent Ineff=
       T
Bank Sta=4978.2,5057.4
XS Rating Curve= 0 ,0
Exp/Cntr=0.3,0.1

Type RM Length L Ch R = 1 ,151458  ,934,934,934
BEGIN DESCRIPTION:
SULPHUR CREEK 164.0
END DESCRIPTION:
XS GIS Cut Line= 4
      2292088.66     13430777.92      2291637.26     13430423.75
      2291296.98     13430486.25      2290326.78     13430970.57
#Sta/Elev= 30
    4205  345.71  4742.1   339.8  4788.5  338.76  4818.8   339.8  4839.3  338.18
    4854  336.56  4876.9  334.11  4962.2  335.11  4981.6  334.77  4988.2  329.59
    4999  326.52  5001.7  326.02    5005  326.52  5022.3  332.77  5046.4   333.7
  5052.8  336.16  5073.3  336.78  5155.8  338.27  5362.7  338.05  5519.3  340.21
  5631.2  339.43  5653.5  338.26  5670.3  335.15  5675.9  336.21  5682.7  334.17
    5715  333.43  5782.2  338.21  5787.8  337.36  5849.3  340.69  6209.1  346.24
#Mann= 7 ,-1 , 0
    4205     .05       0  4742.1      .1       0    4854     .12       0
  4962.2      .1       0    4999     .07       0    5005      .1       0
  5073.3     .05       0
#XS Ineff= 2 , 0
                         5542.61          340.08
Permanent Ineff=
       T       T
Bank Sta=4839.3,5155.8
XS Rating Curve= 0 ,0
Exp/Cntr=0.3,0.1

Type RM Length L Ch R = 1 ,150524  ,598,598,598
BEGIN DESCRIPTION:
Mapping XS 6827378b
END DESCRIPTION:
XS GIS Cut Line= 3
      2292044.31     13430349.75      2291449.89     13429967.63
      2290303.51     13430080.85
#Sta/Elev= 30
    3693  341.95  3858.4  340.19  3931.1  340.43  3952.2  339.68  4018.9  340.34
  4033.7  339.69  4133.8  339.79  4140.7  339.17    4155   340.1  4170.2  340.05
  4388.1  337.84  4662.7  337.19  4733.4  336.82  4743.2   336.7  4823.9  336.37
  4944.5  333.52  4955.4   331.2  4984.6  329.03  4994.7  321.72  5004.5  319.93
  5007.7  320.43  5014.8  323.81  5034.9   329.4  5044.9  329.87  5095.2  336.34
  5105.2  336.75  5145.4     341  5225.8  343.66  5366.5  345.87  5551.6  346.12
#Mann= 4 ,-1 , 0
    3693     .05       0  4662.7      .1       0  4733.4     .07       0
  5105.2     .05       0
Bank Sta=4743.2,5105.2
XS Rating Curve= 0 ,0
Exp/Cntr=0.3,0.1

Type RM Length L Ch R = 1 ,149926  ,615,615,615
BEGIN DESCRIPTION:
SULPHUR CREEK 163.0
END DESCRIPTION:
XS GIS Cut Line= 4
      2292150.48     13428934.47       2291803.7     13429196.32
      2291343.75     13429712.88      2290473.41     13429429.84
#Sta/Elev= 30
  3388.1  345.17  3414.2  343.81  3613.5  335.92  3848.8  337.75  3876.9  335.45
  3890.6  330.84  3912.4  328.33  3919.1  332.28  3990.1  338.24    4047  337.76
  4067.9  340.48  4108.4  335.11  4174.1  337.52  4324.1  337.11  4344.1  336.94
    4667  335.92  4867.6  334.55  4962.3  330.11  4968.9  328.91  4974.2  324.06
  4993.8  320.01  4997.9  317.03  5000.6  316.53  5003.9  317.03  5006.1  320.54
  5025.4  325.02  5081.1  332.56  5101.9  334.75  5183.1   339.2  5429.5  342.69
#Mann= 9 ,-1 , 0
  3388.1     .05       0  3414.2      .1       0  4108.4     .05       0
  4324.1      .1       0  4344.1     .05       0    4667      .1       0
  4997.9     .07       0  5003.9      .1       0  5081.1     .05       0
#XS Ineff= 1 ,-1
 3388.97 4067.89  340.51
Permanent Ineff=
       T
Bank Sta=4867.6,5101.9
XS Rating Curve= 0 ,0
Exp/Cntr=0.3,0.1

Type RM Length L Ch R = 1 ,149311  ,603,603,603
BEGIN DESCRIPTION:
SULPHUR CREEK 162.0
END DESCRIPTION:
XS GIS Cut Line= 6
      2292136.31     13428835.41      2291810.78     13429104.32
      2291464.04     13429153.86      2291074.85     13429090.17
      2290607.82     13429210.47       2290494.2     13429248.33
#Sta/Elev= 30
  4066.1   345.7  4106.3  344.13    4137  342.63  4371.8   333.1  4386.2  335.63
  4435.6   337.6    4552   337.1  4572.2  336.45  4609.9  331.63  4713.7   328.2
  4723.8  324.04  4733.9  328.43    4744   328.9  4751.4  330.99  4827.1  336.64
  4885.5  335.87  4911.9  333.96  4973.3   326.8  4986.9  318.58    4994  317.11
  4996.7  316.61    5000  317.11  5007.1  318.11  5027.4  325.29  5034.6  326.06
  5162.4  333.36    5206  334.12  5508.8  334.23  5644.4  338.19    5835  340.85
#Mann= 6 ,-1 , 0
  4066.1      .1       0  4106.3     .05       0    4137      .1       0
    4994     .07       0    5000      .1       0    5206     .05       0
#XS Ineff= 2 ,-1
  4166.9 4475.25  337.79 4534.65    4843   336.7
Permanent Ineff=
       T       T
Bank Sta=4911.9,5162.4
XS Rating Curve= 0 ,0
Exp/Cntr=0.3,0.1

Type RM Length L Ch R = 1 ,148708  ,580,580,580
BEGIN DESCRIPTION:
SULPHUR CREEK 161.0
END DESCRIPTION:
XS GIS Cut Line= 3
      2291775.36     13428474.55      2290897.94      13428814.2
      2290531.32     13429096.22
#Sta/Elev= 30
  4452.1  340.17  4513.9  337.68  4607.9  335.72  4812.7  334.87  4846.3  334.81
  4878.5  332.88  4885.8  331.33  4891.2  329.09  4899.9  327.96  4933.9  326.29
  4964.3  325.63  4975.7  323.72  4985.7  323.73  4994.9  321.84  4997.2  314.44
    5000  313.94  5003.2  314.44  5007.2  317.95  5017.9  321.47  5024.8  325.16
  5040.5  326.31  5079.3  329.46  5109.2  328.94  5169.1  331.45  5361.3  332.96
  5381.8  333.63  5390.4  332.83  5487.7  333.21    5716  337.67  5855.5  339.37
#Mann= 7 ,-1 , 0
  4452.1     .05       0  4812.7      .1       0  4933.9     .12       0
  4997.2     .07       0  5003.2     .12       0  5040.5      .1       0
  5361.3     .05       0
Bank Sta=4878.5,5169.1
XS Rating Curve= 0 ,0
Exp/Cntr=0.3,0.1

Type RM Length L Ch R = 1 ,148128  ,464,464,464
BEGIN DESCRIPTION:
SULPHUR CREEK 160.0
END DESCRIPTION:
XS GIS Cut Line= 3
      2291637.76     13428196.85      2290837.72     13428296.85
      2290437.69     13428696.89
#Sta/Elev= 30
  4192.9  339.28  4230.7  337.81    4324  335.48  4404.6  334.27  4666.6  334.26
  4757.3  334.03  4800.1  333.69  4804.9  333.31  4888.3  330.45  4898.4  328.91
  4928.6  327.35  4948.8  325.48  4956.3  324.35  4960.6  323.14    4979  319.63
  4991.7   315.5  4993.7  314.61  4996.4  314.11  4999.7  314.61  5002.7  314.61
  5013.3  317.85  5027.5   324.9  5041.6  325.64  5073.2  328.81  5098.2  330.85
  5112.3  330.62  5197.2  332.09    5381  337.91    5480  339.53  5564.9   340.1
#Mann= 7 ,-1 , 0
  4192.9     .05       0  4804.9      .1       0  4960.6     .12       0
  4991.7      .1       0  4993.7     .07       0  4999.7      .1       0
  5073.2     .05       0
Bank Sta=4888.3,5098.2
XS Rating Curve= 0 ,0
Exp/Cntr=0.3,0.1

Type RM Length L Ch R = 1 ,147664  ,710,710,710
BEGIN DESCRIPTION:
SULPHUR CREEK 159.0
END DESCRIPTION:
XS GIS Cut Line= 3
      2291322.53     13427660.77      2290650.27     13427724.45
      2290289.39     13428531.14
#Sta/Elev= 30
  4084.5  335.48  4260.1  333.94  4447.5  333.12  4481.1  334.03  4511.2  333.01
  4546.5  332.91  4734.7  332.18  4853.6  330.22    4900  330.43  4915.8  329.37
  4923.2  327.98  4959.6  325.42  4969.6  323.68  4975.1  323.64  4992.5  316.77
  4995.3  312.26    4998  311.76  5001.3  312.26  5003.8  313.75  5014.4  316.99
  5021.5   322.2  5067.9  326.81  5125.2  326.97  5166.2  328.41  5178.7  329.76
  5233.5  333.23  5287.6  333.38  5408.7  335.18  5484.2  337.04  5643.5  338.74
#Mann= 6 ,-1 , 0
  4084.5     .05       0  4447.5     .08       0  4546.5      .1       0
  4995.3     .07       0  5001.3      .1       0  5125.2     .05       0
Bank Sta=4923.2,5067.9
XS Rating Curve= 0 ,0
Exp/Cntr=0.3,0.1

Type RM Length L Ch R = 1 ,146954  ,510,510,510
BEGIN DESCRIPTION:
SULPHUR CREEK 158.0
END DESCRIPTION:
XS GIS Cut Line= 3
      2289837.71     13426796.82      2290137.72     13427546.85
      2290187.72     13428346.88
#Sta/Elev= 30
  4261.6  340.31  4462.2  328.12  4584.7   325.3  4594.2  315.13  4599.6  314.37
  4617.1  322.29  4657.3  330.01  4809.6  326.93  4812.6  326.64  4839.2  321.82
  4875.5  325.14  4922.7     322  4940.2  320.03  4946.9  313.88  4952.3  317.17
  4971.1  309.43  4976.5  314.98  5003.1  309.29  5005.9  308.79  5009.1  309.29
    5025  319.42  5030.4  312.58  5047.9  319.22  5054.6  319.37    5060   313.4
  5089.5  320.39  5264.5  322.09    5350  327.17  5440.1  331.63    5871  335.98
#Mann= 6 ,-1 , 0
  4261.6      .1       0  4657.3     .08       0  4812.6      .1       0
  5003.1     .07       0  5009.1      .1       0  5264.5     .05       0
#XS Ineff= 1 ,-1
 4350.21 4709.19  331.04
Permanent Ineff=
       T
Bank Sta=4809.6,5350
XS Rating Curve= 0 ,0
Exp/Cntr=0.3,0.1

Type RM Length L Ch R = 1 ,146444  ,495,495,495
BEGIN DESCRIPTION:
SULPHUR CREEK 157.0
END DESCRIPTION:
XS GIS Cut Line= 3
      2289487.71     13426946.82      2289637.72     13427496.85
      2289537.72     13428446.88
#Sta/Elev= 30
  4458.6  337.11  4551.5  334.98  4593.6  333.65  4686.7  332.86  4709.1  331.16
  4728.1  331.53  4806.3  327.88    4818  326.77  4976.9  319.23  4987.3   311.5
  4994.6  309.61  4997.4  309.11  5000.6  309.61  5006.3  311.45  5011.5  311.73
  5026.1  317.67  5031.2  317.67  5038.8  320.26  5082.3  324.49  5139.3  326.74
  5189.6  326.14  5266.3  328.85  5430.9     330  5471.2  331.15  5511.4  330.21
    5622  330.88  5712.5  333.41  5792.9  334.12  5833.1   336.8    5984  338.36
#Mann= 7 ,-1 , 0
  4458.6     .05       0  4551.5      .1       0  4593.6     .08       0
  4806.3      .1       0  4994.6     .07       0  5000.6      .1       0
  5082.3     .05       0
Bank Sta=4818,5139.3
XS Rating Curve= 0 ,0
Exp/Cntr=0.3,0.1

Type RM Length L Ch R = 1 ,145949  ,536,536,536
BEGIN DESCRIPTION:
SULPHUR CREEK 156.0
END DESCRIPTION:
XS GIS Cut Line= 3
      2289287.71     13426946.88      2289137.72     13427596.85
      2289037.72     13428346.86
#Sta/Elev= 30
  4371.7  336.74  4494.8  333.31  4588.7  332.68  4694.9  330.25  4782.2  326.45
  4833.5  323.08  4874.6  322.37  4895.1  323.54  4936.1  320.83  4966.9  315.74
  4977.2  315.54  4987.4  312.34  4994.7   307.3  4997.5   306.8  5000.7   307.3
  5014.8  314.35  5019.9  311.68  5030.4  317.02  5109.4  324.14  5220.4  326.44
    5291  328.86  5321.2  327.75  5432.2  329.75  5456.2  329.08  5492.7  330.72
    5634  332.96  5664.2  335.09  5704.6  334.54  5775.2  337.61  5795.4  337.09
#Mann= 6 ,-1 , 0
  4371.7     .05       0  4588.7     .08       0  4694.9      .1       0
  4994.7     .07       0  5000.7      .1       0  5030.4     .05       0
Bank Sta=4782.2,5220.4
XS Rating Curve= 0 ,0
Exp/Cntr=0.3,0.1

Type RM Length L Ch R = 1 ,145413  ,406,406,406
BEGIN DESCRIPTION:
SULPHUR CREEK 155.0
END DESCRIPTION:
XS GIS Cut Line= 3
       2289037.7     13426946.89      2288637.72     13427696.85
      2288787.73     13428196.88
#Sta/Elev= 30
  4165.1   334.7  4394.3  330.66  4447.3  331.22  4504.4  329.48  4540.8  326.62
  4666.9  326.24  4799.8  327.56  4822.4  327.76  4836.9  326.53  4845.1   324.6
  4858.9  323.93    4941  320.97  4957.3  318.17    4963  318.26    4985  314.14
  4992.4  310.83  4998.2   304.9    5001   304.4  5004.2   304.9  5012.2  312.33
  5017.7  312.33  5031.6  317.05  5069.9  319.35    5109  323.73    5136  325.41
  5169.1  327.31  5317.8  329.47  5416.1  332.91  5487.5  332.82  5537.1  335.37
#Mann= 6 ,-1 , 0
  4165.1     .05       0  4394.3     .08       0  4504.4     .05       0
  4799.8      .1       0  4858.9     .07       0    5136     .05       0
Bank Sta=4845.1,5109
XS Rating Curve= 0 ,0
Exp/Cntr=0.3,0.1

Type RM Length L Ch R = 1 ,145007  ,111,111,111
BEGIN DESCRIPTION:
Mapping XS 095a7359
END DESCRIPTION:
XS GIS Cut Line= 3
      2288144.73      13426670.6      2288201.18     13426844.45
      2288357.23     13428472.81
#Sta/Elev= 30
    4116  331.54  4177.3  329.32  4285.1  330.27  4592.5  327.83  4628.5  328.95
  4682.9  326.08  4823.6  324.12  4873.8  322.91  4954.2  320.13  4974.3  316.21
  4984.3  306.62  4994.1  304.47  5004.4  306.49  5024.5  315.41  5104.9  322.51
    5125  324.63  5151.8  326.26  5156.8  324.53  5362.1  326.34  5367.1  322.22
  5464.8  326.46  5478.4  325.45  5572.4  328.97  5577.4  326.54  5627.2  329.44
  5637.3  328.88  5647.3  325.13  5667.4   330.1  5687.5  332.13  5934.6  335.68
#Mann= 5 ,-1 , 0
    4116     .08       0  4285.1      .1       0  4823.6     .07       0
    5125      .1       0  5478.4     .08       0
Bank Sta=4873.8,5104.9
XS Rating Curve= 0 ,0
Exp/Cntr=0.3,0.1

Type RM Length L Ch R = 1 ,144896  ,484,484,484
BEGIN DESCRIPTION:
SULPHUR CREEK 154.0
END DESCRIPTION:
XS GIS Cut Line= 3
      2288120.87     13426692.36      2288117.69     13426835.47
      2288253.14     13428508.35
#Sta/Elev= 30
  4199.6  332.31  4514.4   331.5  4675.2   331.6  4773.7  329.31  4778.7   331.1
  4835.7  331.13  4875.9  328.87  4895.8  325.84  4900.8  326.48    4906  323.99
  4976.2   314.1  4986.2  307.72    4996  303.67  5006.3  305.96  5016.3  314.36
    5023  314.88    5028  313.53  5036.4  315.62  5106.6  322.06  5116.7   324.8
  5136.7  328.25  5156.8  329.29  5272.3  327.88  5277.3  330.11  5327.3  329.77
  5407.6  331.36  5467.8  329.59  5526.9  331.31  5770.9  333.25  6021.1  337.52
#Mann= 5 ,-1 , 0
  4199.6     .08       0  4514.4      .1       0    4906     .07       0
  5116.7      .1       0  5526.9     .08       0
Bank Sta=4906,5116.7
XS Rating Curve= 0 ,0
Exp/Cntr=0.3,0.1

Type RM Length L Ch R = 1 ,144412  ,460,460,460
BEGIN DESCRIPTION:
SULPHUR CREEK 153.0
END DESCRIPTION:
XS GIS Cut Line= 3
      2288107.32     13426661.15      2287669.81     13427390.33
      2287523.99     13428147.24
#Sta/Elev= 30
  4331.8  332.09  4358.1  332.06  4385.3   329.4    4517  328.69  4803.2  323.75
    4809  324.87  4830.4  321.95  4844.3  322.67  4845.9  322.76  4874.9   320.3
  4904.2  319.14  4925.6  316.32    4947  316.87  4962.5  314.71  4978.1  314.65
  4991.5   303.6  4999.2  301.43  5005.3  302.44  5020.9  317.31  5042.2  313.83
  5049.8  314.17  5079.2  319.32    5085  318.48    5153  323.31  5209.2  324.38
  5229.5  321.77  5249.9  324.54  5599.3  330.07  5699.2  332.89    5953  340.77
#Mann= 7 ,-1 , 0
  4331.8     .08       0    4517      .1       0  4844.3     .12       0
  4874.9     .07       0    5153      .1       0  5599.3     .08       0
  5699.2     .05       0
Bank Sta=4845.9,5153
XS Rating Curve= 0 ,0
Exp/Cntr=0.3,0.1

Type RM Length L Ch R = 1 ,143952  ,593,593,593
BEGIN DESCRIPTION:
SULPHUR CREEK 152.0
END DESCRIPTION:
XS GIS Cut Line= 4
      2288065.68     13426487.53      2287537.87     13426827.83
      2287197.59     13427216.72      2287280.85     13428222.73
#Sta/Elev= 30
  4096.5  330.35  4129.8  331.99  4419.7  327.07  4727.2  326.31  4816.2  322.95
  4837.4  325.64    4844  322.92  4864.3   322.5  4865.9  322.53  4872.5  321.91
  4915.2  320.23  4922.5  318.22  4936.1  318.15  4943.7  314.37  4978.8     312
  4986.4  308.59    4993  308.35  4997.6  302.84  5000.4  302.34  5007.3  303.25
  5014.9   310.4  5085.1  318.02  5104.6  321.63  5142.1  323.82  5191.4  322.41
  5381.9  326.12  5682.9  327.91  5816.2  330.73  6014.6  335.53  6250.7  337.97
#Mann= 7 ,-1 , 0
  4096.5      .1       0  4864.3     .12       0  4865.9     .07       0
  5104.6     .16       0  5104.6      .1       0  5816.2     .08       0
  6014.6      .1       0
Bank Sta=4872.5,5104.6
XS Rating Curve= 0 ,0
Exp/Cntr=0.3,0.1

Type RM Length L Ch R = 1 ,143359  ,444,444,444
BEGIN DESCRIPTION:
SULPHUR CREEK 151.0
END DESCRIPTION:
XS GIS Cut Line= 4
      2287357.31     13426327.83      2287044.81     13426591.72
       2286621.2     13426834.77      2286440.89     13427202.33
#Sta/Elev= 30
  4465.1   331.5  4718.1  324.85    4769  323.06  4776.7  321.75  4832.7   322.2
    4850  320.71  4874.1  319.43  4912.8   313.7  4918.6  315.63  4928.4  312.99
    4963  311.45  4971.8  309.67  4977.6  310.57    4986  305.14  4993.8  301.77
  4996.1   300.9  4998.9   300.4  5002.1   300.9  5009.1  302.71  5020.7  311.82
  5043.7  312.78  5058.1   315.9  5095.5  319.01  5101.3  320.49  5124.4  322.04
    5294  323.04  5388.7  325.21  5487.3  327.75  5567.1  332.92  5771.9  334.83
#Mann= 7 ,-1 , 0
  4465.1     .05       0  4718.1      .1       0    4850     .12       0
  4993.8      .1       0  4996.1     .07       0  5002.1      .1       0
  5388.7     .05       0
Bank Sta=4874.1,5095.5
XS Rating Curve= 0 ,0
Exp/Cntr=0.3,0.1

Type RM Length L Ch R = 1 ,142915  ,559,559,559
BEGIN DESCRIPTION:
SULPHUR CREEK 150.0
END DESCRIPTION:
XS GIS Cut Line= 3
      2287187.75     13426296.85      2286587.72     13426346.85
      2286087.73     13426846.84
#Sta/Elev= 30
  4433.9  328.26  4601.9  324.46  4674.8  323.79  4704.9  321.16  4724.9  323.06
  4765.1  322.64  4775.1  320.93  4795.2  322.27  4865.4  318.41  4915.6  315.59
  4945.7  311.79  4955.7   312.6  4978.3  306.37  4985.8  300.02  4992.9  299.59
  4995.6  299.09  4998.9  299.59  5005.9  303.93  5015.9  305.24    5026  308.67
  5078.4  312.79  5106.7  317.97  5151.8  322.37    5234  320.13    5432  326.95
  5672.4  330.77  5700.7  334.61  5714.8  342.31    5729  346.77  5743.1  347.06
#Mann= 5 ,-1 , 0
  4433.9     .05       0  4601.9      .1       0  4992.9     .07       0
  4998.9      .1       0  5151.8     .05       0
Bank Sta=4865.4,5106.7
XS Rating Curve= 0 ,0
Exp/Cntr=0.3,0.1

Type RM Length L Ch R = 1 ,142356  ,659,659,659
BEGIN DESCRIPTION:
SULPHUR CREEK 149.0
END DESCRIPTION:
XS GIS Cut Line= 3
       2286987.7     13425196.87      2286187.72     13425996.85
      2285687.69     13426396.88
#Sta/Elev= 30
  3869.3  347.22  4307.7  328.46  4505.7  324.16  4641.1  323.42  4760.2   322.4
  4788.5  319.85  4830.9  320.92  4845.1  316.69  4859.2  316.68  4873.4  314.69
  4901.7  316.75  4944.1  316.85  4958.2  312.08  4986.5  305.56  4994.1  299.99
  4996.9  299.49  5000.1  299.99  5003.8  299.99  5014.3  305.54  5028.7  308.59
  5051.1  309.23  5086.3  313.92    5125   316.2  5135.9  316.58  5156.7   318.7
  5220.8  320.29  5320.8  319.33  5467.2  325.95  5634.4  332.69    5641  333.03
#Mann= 7 ,-1 , 0
  3869.3     .05       0  4641.1      .1       0  4994.1     .07       0
  5000.1      .1       0    5125     .05       0  5467.2      .1       0
  5634.4     .05       0
Bank Sta=4944.1,5135.9
XS Rating Curve= 0 ,0
Exp/Cntr=0.3,0.1

Type RM Length L Ch R = 1 ,141697  ,429,429,429
BEGIN DESCRIPTION:
SULPHUR CREEK 148.0
END DESCRIPTION:
XS GIS Cut Line= 3
      2286665.27     13424918.69      2285727.77     13425526.33
      2285397.91     13426081.89
#Sta/Elev= 30
  3739.3  338.89    3783     337  3852.8  334.52  4054.9  327.75  4190.8  326.71
  4272.5  321.69  4293.6  322.89  4299.6  321.05  4314.7  323.43  4423.5  323.95
  4689.7  321.64  4864.7  319.07    4892  315.63  4973.4  307.72  4981.6  305.89
  4993.7  298.13  4996.4  297.63  4999.7  298.13  5008.8  303.16  5024.4  306.99
  5067.3  309.74  5082.9   313.8  5098.5   315.5    5112  317.08  5125.7  319.68
  5242.6  326.55  5264.2  326.08  5345.6  330.82  5368.8   330.4  5502.6  335.32
#Mann= 6 ,-1 , 0
  3739.3      .1       0    3783     .05       0  3852.8      .1       0
  4993.7     .07       0  4999.7      .1       0    5112     .05       0
Bank Sta=4892,5098.5
XS Rating Curve= 0 ,0
Exp/Cntr=0.3,0.1

Type RM Length L Ch R = 1 ,141268  ,485,485,485
BEGIN DESCRIPTION:
SULPHUR CREEK 147.0
END DESCRIPTION:
XS GIS Cut Line= 2
      2285432.63      13424519.4      2285259.26     13425923.73
#Sta/Elev= 30
  4129.7  343.44  4460.1  327.11    4510  325.91  4560.4  323.16    4772  318.42
  4811.8  315.21  4812.3  315.17  4872.8  311.39    4903  311.57  4981.9   305.7
  4983.6  305.52  4993.7  299.26  5000.7  296.65  5003.5  296.15  5006.7  296.65
  5013.8  301.44  5027.8  305.99  5054.1  307.86  5084.4  312.43  5134.7  315.18
    5165  317.98  5215.3  320.87  5265.7  321.92  5276.2  323.55  5346.3  326.93
  5416.9  328.77  5447.1  330.93  5497.5   331.6  5537.8  333.14  5544.7  334.38
#Mann= 5 ,-1 , 0
  4129.7     .05       0  4811.8      .1       0  4981.9     .05       0
  5000.7     .03       0  5006.7     .05       0
Bank Sta=4812.3,5134.7
XS Rating Curve= 0 ,0
Exp/Cntr=0.3,0.1

Type RM Length L Ch R = 1 ,140783  ,532,532,532
BEGIN DESCRIPTION:
SULPHUR CREEK 146.0
END DESCRIPTION:
XS GIS Cut Line= 3
      2285237.72     13424446.85      2284887.72     13425196.85
      2285037.71     13425846.82
#Sta/Elev= 30
  4171.5  345.99  4208.5  344.45  4215.6  343.15    4315   337.4  4345.7  334.54
  4488.4  327.01  4539.6     326  4601.9  322.95  4813.6  318.68  4865.1  318.09
    4900  314.63  4932.9  307.57  4990.5  302.53  4993.4  294.53  4996.1  294.03
  4999.4  294.53  5001.7  294.53    5018  301.47  5060.7  300.24    5071  304.19
  5081.3  306.51  5101.8  310.74  5114.1  311.72  5122.3  314.15  5296.8  320.01
  5368.6  321.02  5399.4  322.33  5409.7  323.92  5481.5  324.54  5666.2  331.44
#Mann= 5 ,-1 , 0
  4171.5     .05       0  4813.6      .1       0  4993.4     .07       0
  4999.4      .1       0  5114.1     .05       0
Bank Sta=4900,5122.3
XS Rating Curve= 0 ,0
Exp/Cntr=0.3,0.1

Type RM Length L Ch R = 1 ,140251  ,578,578,578
BEGIN DESCRIPTION:
SULPHUR CREEK 145.0
END DESCRIPTION:
XS GIS Cut Line= 3
      2284737.71     13424596.86      2284387.72     13425046.85
      2284087.69     13425396.89
#Sta/Elev= 30
  4420.4  328.63  4427.6  327.48  4483.7  325.64  4506.4  323.37  4676.5  317.13
  4841.8  318.26  4862.9  317.39    4890  314.24  4904.5  312.74  4912.7  310.49
  4947.9  305.82  4976.9  304.73  4983.5  301.69  4987.3  295.11  4994.6  294.78
  4997.4  294.28  5000.6  294.78  5004.2   295.1  5011.9  300.21  5026.1  301.16
    5047  306.82  5061.3  307.91  5082.7  312.33  5104.1  314.22    5110  315.04
  5124.9  315.13  5139.2  316.98  5196.3  319.32  5231.4  322.06  5451.5  329.85
#Mann= 6 ,-1 , 0
  4420.4     .05       0  4841.8     .12       0  4983.5      .1       0
  4994.6     .07       0  5000.6      .1       0    5110     .05       0
Bank Sta=4890,5104.1
XS Rating Curve= 0 ,0
Exp/Cntr=0.3,0.1

Type RM Length L Ch R = 1 ,139673  ,548,548,548
BEGIN DESCRIPTION:
SULPHUR CREEK 144.0
END DESCRIPTION:
XS GIS Cut Line= 3
      2284287.71     13423896.87      2283937.72     13424696.85
      2283887.72     13425096.85
#Sta/Elev= 30
  4126.7  342.79  4508.3  320.43    4596  317.65    4705  315.91    4727  316.08
  4816.3  312.11  4857.6   310.4  4919.1     305  4933.2  303.78  4938.7  304.38
  4945.3  302.69  4962.1  303.48  4967.5  301.31  4978.1  301.28  4985.5   298.9
  4994.2  294.06  4996.9  293.56  5000.2  294.06    5010  294.48    5020  300.08
  5037.7   303.8  5042.7  309.12  5063.6  312.53  5070.4  312.48  5080.5  314.57
  5123.3   318.9  5198.9  322.46  5211.5  323.94  5264.5  324.51    5403  326.35
#Mann= 7 ,-1 , 0
  4126.7     .05       0    4705      .1       0  4919.1     .12       0
  4994.2     .07       0  5000.2     .12       0  5063.6      .1       0
  5264.5     .05       0
Bank Sta=4816.3,5070.4
XS Rating Curve= 0 ,0
Exp/Cntr=0.3,0.1

Type RM Length L Ch R = 1 ,139125  ,446,446,446
BEGIN DESCRIPTION:
SULPHUR CREEK 143.0
END DESCRIPTION:
XS GIS Cut Line= 3
      2283837.73     13423946.85      2283587.72     13424296.85
      2283387.74     13424646.82
#Sta/Elev= 30
  4566.9  324.24  4574.3  323.12  4595.2  322.89  4630.8  320.32  4710.7  317.17
  4853.2  314.33  4861.8  312.38  4874.1  312.25  4888.9  310.66  4905.4   308.3
  4939.3  303.81  4968.8  302.96  4974.9  301.22  4983.5  302.19    4991  293.65
  4993.7  293.15    4997  293.65  5010.7  295.05  5020.1  297.33  5032.3  301.95
  5042.4  303.72    5064  305.39  5069.7  308.29  5085.6  307.97  5100.7   311.1
  5109.4  312.99  5215.9  320.58  5282.1  321.93  5395.7  324.54  5400.1  324.62
#Mann= 7 ,-1 , 0
  4566.9     .05       0  4905.4     .12       0    4991     .07       0
    4997     .12       0  5109.4      .1       0  5282.1     .05       0
  5395.7      .1       0
Bank Sta=4888.9,5100.7
XS Rating Curve= 0 ,0
Exp/Cntr=0.3,0.1

Type RM Length L Ch R = 1 ,138679  ,492,492,492
BEGIN DESCRIPTION:
SULPHUR CREEK 142.0
END DESCRIPTION:
XS GIS Cut Line= 2
      2283687.71     13423446.86      2282715.62     13424701.68
#Sta/Elev= 30
  4271.4  340.88  4278.6  338.83  4313.9  336.06  4549.7  322.74  4585.6  321.85
    4600  325.08  4612.9  323.62  4620.9  320.25  4627.2  319.71  4726.8  315.71
  4863.5  313.46  4869.8  314.58  4905.1  310.78  4940.5  304.11  4977.6  300.08
  4995.4  292.53  4998.1  292.03  5001.4  292.53  5005.1  293.47  5012.9  299.65
  5019.2     301  5118.9   310.3  5176.7  315.92    5224  317.65  5241.2  318.02
  5475.5  323.07  5724.5  324.18  5729.2   324.1  5825.3  324.58  5858.7   324.7
#Mann= 9 ,-1 , 0
  4271.4     .05       0  4940.5     .12       0  4995.4     .07       0
  5001.4     .12       0    5224      .1       0  5241.2     .05       0
  5724.5      .1       0  5729.2     .05       0  5825.3      .1       0
Bank Sta=4905.1,5118.9
XS Rating Curve= 0 ,0
Exp/Cntr=0.3,0.1

Type RM Length L Ch R = 1 ,138187  ,802,802,802
BEGIN DESCRIPTION:
SULPHUR CREEK 141.0
END DESCRIPTION:
XS GIS Cut Line= 3
       2283132.3     13422896.08      2282949.99     13423590.57
      2282429.14     13424328.44
#Sta/Elev= 30
  4138.9  337.99  4408.1  323.94  4677.3  313.57  4725.9  312.15  4822.1  313.35
  4841.9  310.28  4856.9   310.6    4864  308.54  4870.1  313.21  4884.9  309.16
  4895.7  310.39  4913.6  309.11  4920.6  304.96  4926.7  308.73  4935.4  307.57
  4941.5  309.86  4956.3  308.98  4971.1  300.98    4992  294.82  4996.3  291.41
    4999  290.91  5002.3  291.41  5021.6  300.33  5083.8  302.52  5149.6   308.6
  5207.3  315.06  5351.6  319.66  5452.1  321.02  5530.1  320.09  5760.1  324.13
#Mann= 5 ,-1 , 0
  4138.9     .05       0  4895.7      .1       0  4996.3     .07       0
  5002.3      .1       0  5083.8     .05       0
Bank Sta=4956.3,5149.6
XS Rating Curve= 0 ,0
Exp/Cntr=0.3,0.1

Type RM Length L Ch R = 1 ,137385  ,734,734,734
BEGIN DESCRIPTION:
SULPHUR CREEK 140.0
END DESCRIPTION:
XS GIS Cut Line= 4
      2282837.17     13422696.46      2282298.95     13423139.18
      2282021.17     13423538.49      2281969.09     13424146.13
#Sta/Elev= 30
  4088.6   338.8  4159.6  336.47  4422.9  320.64    4557  314.18  4635.2  312.64
  4770.8     315  4828.4  312.04  4864.5  307.03    4906  302.64  4965.4  298.86
  4977.6  298.94  4986.4  293.58  4998.2  290.42    5001  289.92  5004.2  290.42
  5007.3  290.99  5014.1  297.52  5028.2  298.33  5060.4  305.61    5064  306.83
  5072.8  307.44  5123.4  313.02  5129.5  314.57  5180.1  315.81  5230.8  315.39
  5481.1  317.88  5492.1  318.65  5600.8   319.1  5838.3  323.69  5881.8   323.8
#Mann= 5 ,-1 , 0
  4088.6     .05       0  4864.5      .1       0  4998.2     .07       0
  5004.2      .1       0  5060.4     .05       0
Bank Sta=4864.5,5072.8
XS Rating Curve= 0 ,0
Exp/Cntr=0.3,0.1

Type RM Length L Ch R = 1 ,136651  ,690,690,690
BEGIN DESCRIPTION:
SULPHUR CREEK 139.0
END DESCRIPTION:
XS GIS Cut Line= 4
      2282672.26     13422514.18      2282012.49     13422557.58
      2281656.59      13422861.4      2281752.07     13423599.22
#Sta/Elev= 30
  4077.5  332.59  4643.3  316.77  4791.1  309.67  4848.3  305.78  4932.8   298.5
  4954.8  297.02  4968.5  299.23  4975.7   298.7  4982.3  297.39    4990  293.27
  4996.5  291.73  5001.2  288.53    5004  288.03  5007.2  288.53  5018.5  294.36
  5025.1  294.93  5032.8  297.72  5036.6  297.34  5074.5   299.3  5096.5  304.57
  5117.3  306.77    5125  309.91  5152.6  313.48  5207.2   314.8  5235.5  315.01
  5249.4  315.38  5445.5  315.01  5625.6  313.94  5736.9  315.02  5950.6  317.55
#Mann= 11 ,-1 , 0
  4077.5     .05       0  4791.1      .1       0  4932.8     .12       0
  5001.2     .07       0  5007.2     .12       0  5036.6      .1       0
  5207.2     .05       0  5235.5      .1       0  5249.4     .05       0
  5445.5      .1       0  5736.9     .05       0
Bank Sta=4848.3,5117.3
XS Rating Curve= 0 ,0
Exp/Cntr=0.3,0.1

Type RM Length L Ch R = 1 ,135961  ,562,562,562
BEGIN DESCRIPTION:
SULPHUR CREEK 138.0
END DESCRIPTION:
XS GIS Cut Line= 3
      2281873.63     13421663.45      2281179.16     13422479.46
      2280710.43     13423156.51
#Sta/Elev= 30
  4198.7  331.81  4475.1  319.33  4623.4  314.04    4787  309.65  4864.9  310.53
  4900.1  305.57  4904.9  304.93  4922.1  301.53  4942.9  299.31  4950.6  297.09
  4971.5  294.92  4985.7  287.56  4989.3  286.91  4992.1  286.41  4995.3  286.91
    5000  288.03  5014.3  296.14  5020.9   297.2  5049.4  296.49  5084.6  299.41
  5135.1   305.5    5144  305.83  5198.8  310.41  5253.2  311.97  5291.4  311.82
    5413  315.84  5505.4  316.34  5611.4  315.77  5772.6  314.56  6093.7  316.94
#Mann= 8 ,-1 , 0
  4198.7     .05       0  4904.9     .12       0  4989.3     .07       0
  4995.3     .12       0    5144      .1       0  5253.2     .05       0
  5505.4      .1       0  5611.4     .05       0
Bank Sta=4900.1,5135.1
XS Rating Curve= 0 ,0
Exp/Cntr=0.3,0.1

Type RM Length L Ch R = 1 ,135399  ,433,433,433
BEGIN DESCRIPTION:
SULPHUR CREEK 137.0
END DESCRIPTION:
XS GIS Cut Line= 3
      2281637.73     13421446.85      2280837.72     13422046.85
      2280487.74     13422246.84
#Sta/Elev= 30
  4012.2  334.03  4240.3  322.32  4590.3  307.63  4725.8  309.43  4780.9   307.6
  4875.8  305.46  4890.3  304.53  4898.7  302.66  4919.5  297.26  4954.9  296.54
  4969.5  295.07  4975.8  289.33  4984.1  288.43  4987.3  287.06  4990.1  286.56
  4993.3  287.06  4998.7   287.5  5005.2  291.79  5009.1  294.95  5035.2  295.19
  5057.6  303.76  5063.3  301.95  5079.2  305.58  5084.9  302.44  5092.8  302.79
  5150.4  310.65  5187.1  311.58    5203   313.5  5366.6   316.4  5415.3   316.6
#Mann= 6 ,-1 , 0
  4012.2     .05       0  4780.9     .12       0  4987.3     .07       0
  4993.3     .12       0  5005.2      .1       0  5366.6     .05       0
Bank Sta=4898.7,5057.6
XS Rating Curve= 0 ,0
Exp/Cntr=0.3,0.1

Type RM Length L Ch R = 1 ,134966  ,548,548,548
BEGIN DESCRIPTION:
SULPHUR CREEK 136.0
END DESCRIPTION:
XS GIS Cut Line= 3
       2281410.4      13421348.7      2280249.42     13421863.47
      2279778.46     13421934.66
#Sta/Elev= 30
  4067.6  328.48  4171.6  323.86  4324.8  316.86  4394.7  311.19  4486.2  306.14
  4545.3  305.03  4568.5   302.8  4628.4  303.02  4667.1  305.92  4703.8  304.93
  4742.4  304.64  4788.9  300.64    4841  299.58  4864.2  296.25  4968.3  296.52
  4991.5  292.54  5000.3   287.4  5006.3  287.28  5009.1  286.78  5012.3  287.28
  5014.8  291.51  5037.5  297.81  5044.1  301.98    5055   309.4  5061.4  311.17
  5120.7  313.44  5153.5  311.78  5258.5  314.96    5582  315.35  5813.9  317.71
#Mann= 6 ,-1 , 0
  4067.6     .05       0  4171.6      .1       0  4703.8     .12       0
  5006.3     .07       0  5012.3     .12       0  5037.5     .05       0
Bank Sta=4788.9,5044.1
XS Rating Curve= 0 ,0
Exp/Cntr=0.3,0.1

Type RM Length L Ch R = 1 ,134418  ,646,646,646
BEGIN DESCRIPTION:
SULPHUR CREEK 135.0
END DESCRIPTION:
XS GIS Cut Line= 3
      2280937.72     13420796.85      2280687.72     13421146.85
      2279687.73     13421796.85
#Sta/Elev= 30
  4443.9  323.93  4579.1  321.17  4625.7  314.26  4652.8  307.73 4661.82  300.59
  4679.9   293.2  4765.9  294.43    4788  290.45  4810.1  294.59  4902.7  294.13
  4917.8  288.54  4923.8  291.84    4933  288.87  4938.9  293.52  4966.2   286.5
    4969     286  4972.2   286.5  4975.2  289.54  5005.2   286.8  5011.4  292.12
  5017.4  287.15  5026.5  290.89  5032.5  287.92  5047.7  298.73  5053.6  295.58
 5058.64   300.4  5071.6  299.31  5083.9  309.67  5171.6  308.38  6066.7  319.01
#Mann= 6 ,-1 , 0
  4443.9     .16       0  4625.7     .12       0  4966.2     .07       0
  4972.2     .12       0  5071.6      .1       0  5171.6     .05       0
#XS Ineff= 1 ,-1
  5097.6 5489.67  310.69
Permanent Ineff=
       T
Bank Sta=4661.82,5058.64
XS Rating Curve= 0 ,0
Exp/Cntr=0.3,0.1

Type RM Length L Ch R = 1 ,133772  ,554,554,554
BEGIN DESCRIPTION:
SULPHUR CREEK 134.0
END DESCRIPTION:
XS GIS Cut Line= 3
      2280887.71     13420696.86      2280487.72     13420746.85
      2279637.69     13421696.89
#Sta/Elev= 30
    4634  327.74  4772.1  322.57  4871.5  315.85    4896  310.83  4906.1  303.96
 4909.89   299.4  4913.6  296.39  4918.7   294.1  4946.4  294.58  4976.6  292.74
  4986.7  290.18  4996.3  284.47  4999.1  283.97  5002.3  284.47  5006.9  285.42
  5016.9  290.87    5027  293.79  5039.8  294.99  5058.4  295.92  5086.8  294.01
    5101  294.35  5171.3  299.52  5211.8  303.61  5284.9  308.52  5405.3  306.84
  5533.2  307.33  5625.1     309  5752.2  313.32  6049.8  312.91  6311.9  318.34
#Mann= 7 ,-1 , 0
    4634     .05       0  4772.1     .16       0  4871.5     .12       0
  4996.3     .07       0  5002.3     .12       0  5039.8      .1       0
  5211.8     .05       0
Bank Sta=4909.89,5171.3
XS Rating Curve= 0 ,0
Exp/Cntr=0.3,0.1

Type RM Length L Ch R = 1 ,133218  ,481,481,481
BEGIN DESCRIPTION:
SULPHUR CREEK 133.0
END DESCRIPTION:
XS GIS Cut Line= 3
      2279937.71     13419646.81      2280087.72     13420396.85
      2279537.74     13421646.81
#Sta/Elev= 30
  4211.5   325.1  4368.6  316.69  4405.3  314.67  4456.3  307.16  4486.9  306.58
  4599.1  295.41  4721.4  294.52  4741.8  295.51  4772.4  300.71  4792.8  302.27
  4843.8  298.39  4853.1  299.22  4864.2  297.11  4935.6  291.12  4979.1  293.14
  4995.2  285.95    4998  285.45  5001.2  285.95  5008.3  285.98  5014.1  290.43
  5020.1  292.76  5037.5  292.34  5074.7  297.84  5096.6  300.32  5136.3  301.55
  5227.7  307.63  5432.8  305.61  5795.8  311.05  5970.6  310.75    6342   318.3
#Mann= 6 ,-1 , 0
  4211.5      .1       0  4368.6     .05       0  4853.1     .12       0
  4995.2     .07       0  5001.2     .12       0  5008.3     .05       0
#XS Ineff= 2 ,-1
 4318.25 4795.62  301.96 5251.77 5654.88  307.88
Permanent Ineff=
       T       T
Bank Sta=4864.2,5074.7
XS Rating Curve= 0 ,0
Exp/Cntr=0.3,0.1
