HEC-RAS study SULPHUR CREEK.prj: SULPHUR CREEK Base Level Engineering

--- SULPHUR CREEK.g01 (geometry) --- (continued)

Type RM Length L Ch R = 1 ,132737  ,407,407,407
BEGIN DESCRIPTION:
SULPHUR CREEK 132.0
END DESCRIPTION:
XS GIS Cut Line= 4
      2279822.59     13419626.44       2279808.7     13419918.11
      2279586.48     13420334.77      2279482.31     13421529.22
#Sta/Elev= 30
  4455.2   326.7  4604.2   319.3  4685.9     315  4715.9   311.7  4749.3  309.54
  4783.3   305.4  4821.5  302.22  4827.2   300.9  4852.4  298.25  4893.1  294.74
  4909.4  292.48  4917.8  292.42  4975.3  291.74  4983.8  290.72  4994.2  287.05
    4997  286.55  5000.2  287.05    5007  287.55  5025.3  289.29  5117.6  297.44
  5131.1  297.73  5211.1  304.01  5271.7  306.79  5372.1  307.38  5512.6  305.09
  5562.8  305.14  5924.2  308.93  6084.8  309.42  6299.6  312.95  6418.4  315.94
#Mann= 8 ,-1 , 0
  4455.2      .1       0  4604.2     .05       0  4852.4      .1       0
  4917.8     .12       0  4994.2     .07       0  5000.2     .12       0
    5007      .1       0  5025.3     .05       0
#XS Ineff= 2 , 0
                         5360.17          307.73
Permanent Ineff=
       T       T
Bank Sta=4852.4,5131.1
XS Rating Curve= 0 ,0
Exp/Cntr=0.3,0.1

Type RM Length L Ch R = 1 ,132330  ,571,571,571
BEGIN DESCRIPTION:
SULPHUR CREEK 131.0
END DESCRIPTION:
XS GIS Cut Line= 3
      2279537.71     13419596.88      2279337.72     13419946.85
      2279387.72     13421496.86
#Sta/Elev= 30
  4602.9  325.26  4764.1  316.91  4777.8  317.12  4836.8  313.21  4844.7  308.05
  4858.4  303.44  4890.1  297.85  4895.9  295.93  4925.4  293.04  4933.3  290.94
  4948.4     290  4976.5  292.26  4995.1  285.68  4997.8  285.18  5001.1  285.68
  5003.1  287.59    5016  288.04    5026  292.48    5036  293.16    5086   291.7
  5115.1  293.02  5176.1  296.89  5296.1  305.54  5326.2  304.78  5506.2  306.45
  5646.3  304.61  5766.4  306.54  6116.6  307.81  6256.6  309.55  6556.8  315.74
#Mann= 4 ,-1 , 0
  4602.9      .1       0  4995.1     .07       0  5001.1      .1       0
  5115.1     .05       0
Bank Sta=4895.9,5176.1
XS Rating Curve= 0 ,0
Exp/Cntr=0.3,0.1

Type RM Length L Ch R = 1 ,131759  ,515,515,515
BEGIN DESCRIPTION:
SULPHUR CREEK 130.0
END DESCRIPTION:
XS GIS Cut Line= 3
      2279087.71     13419246.87      2278887.72     13419596.85
      2278401.35     13420673.83
#Sta/Elev= 30
    4569   330.8  4663.3   326.9  4679.1  324.66  4759.7  321.43  4807.7  317.67
    4921  313.17  4926.7  312.16  4936.8  306.43  4942.6  309.29  4949.1  302.15
  4958.4  298.68  4964.2  303.14  4969.2  293.82  4972.1  293.82    4994  285.46
    5001  285.17  5003.8  284.67    5007  285.17    5016  292.11  5078.9  289.85
  5107.5  291.33  5235.4  288.41  5303.4   290.9  5349.7   294.5    5411  302.61
  5424.5  301.42  5476.8  305.84  5608.5  303.42    5645  304.41  6153.8  304.47
#Mann= 5 ,-1 , 0
    4569     .08       0  4807.7      .1       0    5001     .07       0
    5007      .1       0    5645     .05       0
Bank Sta=4972.1,5349.7
XS Rating Curve= 0 ,0
Exp/Cntr=0.3,0.1

Type RM Length L Ch R = 1 ,131244  ,577,577,577
BEGIN DESCRIPTION:
SULPHUR CREEK 129.0
END DESCRIPTION:
XS GIS Cut Line= 3
      2278687.74     13419196.84      2278387.72     13419496.85
      2277982.33     13420469.79
#Sta/Elev= 30
  4577.6  321.42  4789.8  309.96  4846.3  302.66  4860.5  305.39  4874.6   301.7
  4888.7  304.53  4902.9  303.55    4917  293.82  4931.2  291.09  4945.3  293.11
  4954.9  291.39  4973.6   292.8  4984.7  285.62  4987.5  285.12  4990.7  285.62
  5004.6  285.67  5011.1  290.25  5023.6  291.17  5180.9  287.72  5207.7  286.21
  5276.5   287.9  5353.4  290.66  5370.2  294.36  5377.3  299.28  5382.7  298.07
  5454.2  304.93  5749.4  302.19  5791.1  304.28  5843.2  303.49  6055.9  303.99
#Mann= 6 ,-1 , 0
  4577.6      .1       0  4954.9     .12       0  4984.7     .07       0
  4990.7     .12       0  5180.9      .1       0  5843.2     .05       0
Bank Sta=4917,5370.2
XS Rating Curve= 0 ,0
Exp/Cntr=0.3,0.1

Type RM Length L Ch R = 1 ,130667  ,562,562,562
BEGIN DESCRIPTION:
SULPHUR CREEK 128.0
END DESCRIPTION:
XS GIS Cut Line= 3
       2278187.7     13418996.89      2277937.72     13419546.85
      2277628.84     13420288.17
#Sta/Elev= 30
  4372.6  313.38  4394.5  312.85  4416.5  309.06  4484.6  306.26  4507.7  302.89
  4582.4  297.08  4713.1  293.75  4903.7  288.06  4944.9  287.47  4979.4  289.79
  4985.9  284.85  4995.4  282.07  4998.1  281.57  5001.4  282.07  5009.2  287.12
  5015.2   287.9  5068.3  287.46  5081.1  288.72  5128.4  293.36  5150.6  294.83
    5169  294.01  5174.4  295.36    5215  295.59  5227.5  296.95  5269.2   297.2
  5328.3  302.44  5550.9  304.03  5712.8  301.37  5753.7  302.09  5779.8  302.04
#Mann= 6 ,-1 , 0
  4372.6     .05       0  4903.7     .12       0  4995.4     .07       0
  5001.4     .12       0  5081.1      .1       0  5753.7     .05       0
Bank Sta=4713.1,5128.4
XS Rating Curve= 0 ,0
Exp/Cntr=0.3,0.1

Type RM Length L Ch R = 1 ,130105  ,540,540,540
BEGIN DESCRIPTION:
SULPHUR CREEK 127.0
END DESCRIPTION:
XS GIS Cut Line= 3
      2277787.71     13418696.88      2277387.72     13419446.85
      2277203.63     13420183.22
#Sta/Elev= 30
  4141.1  316.14  4186.4   314.4  4275.3  306.52  4341.2  302.24  4489.2  296.59
  4555.1  296.21  4560.8  297.31    4577  297.35    4599  296.31  4642.9  291.61
  4696.4  290.73  4753.1  287.97  4864.7  287.28  4911.4  286.69  4955.3  288.62
  4977.3  288.46  4982.9  288.02  4985.2  281.98    4988  281.48  4991.2  281.98
  5001.4   282.1  5009.1  287.79  5032.3  286.39  5042.3  287.26  5050.3  291.26
  5063.2  293.89  5083.8  295.64  5302.9  300.29  5591.5  300.24  5750.1  301.86
#Mann= 5 ,-1 , 0
  4141.1     .05       0  4864.7     .12       0  4985.2     .07       0
  4991.2     .12       0  5042.3      .1       0
Bank Sta=4642.9,5050.3
XS Rating Curve= 0 ,0
Exp/Cntr=0.3,0.1

Type RM Length L Ch R = 1 ,129565  ,1843,1843,1843
BEGIN DESCRIPTION:
SULPHUR CREEK 126.0
END DESCRIPTION:
XS GIS Cut Line= 3
      2277137.74     13418646.82      2276887.72     13419246.85
      2276795.06     13420358.76
#Sta/Elev= 30
  4334.9  311.66  4389.1  309.14  4562.4  305.94  4633.4   299.3  4768.8  295.31
  4811.1  290.42  4823.8  289.74  4840.3  286.97  4887.4  284.84  4938.4  286.43
  4970.3  286.43  4975.7  284.21    4992  282.39  4994.7  281.89    4998  282.39
    5015  287.81  5095.3  286.22  5145.5  287.91  5255.9  285.37  5306.1  290.09
  5486.7  290.56  5556.9  289.02  5677.3  291.99  5757.6  296.04  5787.7  299.31
    5858   293.5  5908.1  299.84  5928.2  300.67  6072.6  299.71  6100.7  299.63
#Mann= 6 ,-1 , 0
  4334.9     .05       0  4823.8     .12       0  4938.4      .1       0
    4992     .07       0    4998      .1       0  6072.6     .05       0
Bank Sta=4811.1,5306.1
XS Rating Curve= 0 ,0
Exp/Cntr=0.3,0.1

Type RM Length L Ch R = 1 ,127722  ,1290,1290,1290
BEGIN DESCRIPTION:
SULPHUR CREEK 125.0
END DESCRIPTION:
XS GIS Cut Line= 4
      2276804.18     13418104.42      2276125.75     13419564.81
      2275781.23     13420539.72      2276092.34     13421411.71
#Sta/Elev= 30
  2611.7  324.41    2708  321.12  3280.6  301.25  3816.3  296.98  4186.3  299.67
  4348.6  293.69  4431.2   293.9  4534.7  289.38  4552.9  289.36    4659  284.05
  4733.8  283.48  4741.8  283.16  4845.4  283.77  4927.1  283.54    4951  280.88
  4956.3  282.94  4973.6  278.86  4976.4  278.36  4979.6  278.86  4981.9  282.29
  4987.8  279.07  5038.5  283.68  5043.8  281.32 5056.82   289.9  5069.4  299.34
  5074.7  292.14  5093.8  298.96  5150.3  299.14  5624.5  301.69  6181.8   316.2
#Mann= 12 ,-1 , 0
  2611.7      .1       0    2708     .05       0  4186.3      .1       0
  4431.2     .12       0  4534.7      .1       0  4733.8     .12       0
  4741.8      .1       0  4845.4     .12       0  4927.1      .1       0
  4973.6     .07       0  4979.6      .1       0  5150.3     .05       0
#XS Ineff= 2 , 0
         4135.08  300.28
Permanent Ineff=
       T       T
Bank Sta=4552.9,5056.82
XS Rating Curve= 0 ,0
Exp/Cntr=0.3,0.1

Type RM Length L Ch R = 1 ,126432  ,1743,1743,1743
BEGIN DESCRIPTION:
SULPHUR CREEK 124.0
END DESCRIPTION:
XS GIS Cut Line= 4
      2276264.44     13418051.78      2275457.14     13418898.14
      2275274.85     13420004.91      2276042.49     13421722.34
#Sta/Elev= 30
  3327.5  307.99  3639.8  297.13  3866.3  294.25  4163.5  296.53  4707.3  296.45
  4861.2   294.2  4870.8  293.46    4881  289.12  4901.2  284.23  4982.3  279.89
  4999.6  276.06  5002.3  275.56  5005.6  276.06  5012.1  279.67  5022.8  280.96
  5173.4   281.5  5296.5   281.6  5316.7  283.85  5328.1  288.83  5362.3  291.46
  5573.9  292.36  5712.8  297.16  5730.5  300.51  5741.5   297.5  6129.3  297.03
  6168.6  294.44  6213.5  297.01  6628.7  303.71    7023  314.75    7500  319.74
#Mann= 9 ,-1 , 0
  3327.5     .05       0  4707.3      .1       0  4861.2     .12       0
  4999.6     .07       0  5005.6     .12       0  5173.4      .1       0
  5362.3     .12       0  5573.9      .1       0  6213.5     .05       0
#XS Ineff= 2 , 0
                         5729.84          300.65
Permanent Ineff=
       T       T
Bank Sta=4881,5328.1
XS Rating Curve= 0 ,0
Exp/Cntr=0.3,0.1

Type RM Length L Ch R = 1 ,124689  ,776,776,776
BEGIN DESCRIPTION:
SULPHUR CREEK 123.0
END DESCRIPTION:
XS GIS Cut Line= 3
      2275037.71     13418646.88      2274387.72     13420096.85
      2274437.72     13420496.85
#Sta/Elev= 30
  3431.4  297.27  3434.7  297.27  3733.8     296  3857.8  295.38  4007.9  295.99
  4670.6  294.19  4716.8  289.36  4734.6  287.23  4809.6  284.36  4838.3  280.25
  4890.2  280.93  4954.2  277.15  4982.9  277.52  4988.4  277.08  4995.5  272.23
  4998.2  271.73  5001.5  272.23  5011.5   274.8  5017.7  280.37  5022.9  280.37
 5032.67  287.12  5040.5     293  5050.6  294.63  5127.4  294.17  5138.8  294.72
  5143.8  290.21  5151.4  293.66  5161.5  294.95  5196.9  296.21  5423.5  297.85
#Mann= 10 ,-1 , 0
  3431.4      .1       0  3434.7     .08       0  3733.8      .1       0
  3857.8     .08       0  4007.9      .1       0  4716.8     .12       0
  4995.5     .07       0  5001.5     .12       0  5127.4      .1       0
  5196.9     .05       0
#XS Ineff= 2 , 0
         3958.27   297.2
Permanent Ineff=
       T       T
Bank Sta=4734.6,5032.67
XS Rating Curve= 0 ,0
Exp/Cntr=0.3,0.1

Type RM Length L Ch R = 1 ,123913  ,2050,2050,2050
BEGIN DESCRIPTION:
Mapping XS b80bc35e
END DESCRIPTION:
XS GIS Cut Line= 4
      2274980.74     13418549.28      2274690.13     13418945.45
      2273683.18     13419674.62      2273813.92     13420402.71
#Sta/Elev= 30
  3690.7  297.07    3757  296.13  4242.3  293.53  4665.3   293.9  4692.4  292.81
  4715.6  288.19  4736.5   290.7  4742.7  293.13  4778.2   289.6  4785.8  290.88
  4822.3  284.23  4893.5  276.54  4979.3  275.06  4987.5  270.76  4997.2  270.18
  4999.9  269.68  5003.2  270.18  5008.7  274.88  5014.9  275.24  5023.4  278.28
  5030.1  277.51  5036.9  285.51  5044.3  286.83  5050.4  290.94    5059  290.54
  5065.1  294.19  5205.1  294.45  5872.4  295.43  5931.2  294.02    6165  295.26
#Mann= 7 ,-1 , 0
  3690.7     .08       0    3757      .1       0  4785.8     .12       0
  4997.2     .07       0  5003.2     .12       0  5030.1      .1       0
  5205.1     .05       0
Bank Sta=4822.3,5036.9
XS Rating Curve= 0 ,0
Exp/Cntr=0.3,0.1

Type RM Length L Ch R = 1 ,121863  ,1051,1051,1051
BEGIN DESCRIPTION:
SULPHUR CREEK 122.0
END DESCRIPTION:
XS GIS Cut Line= 4
      2274187.71     13416646.89      2273803.49     13417478.87
       2273661.8     13418078.42      2273683.54     13419103.01
#Sta/Elev= 30
  3950.1  298.58  3951.1  298.58  4357.6  296.54  4594.5  292.38  4628.7  290.73
  4698.6   290.8  4823.2  289.15  4913.1  290.08  4959.4  290.86  4967.2   288.8
 4975.57  281.43  4977.5  278.56 4983.52  281.16  4987.7   272.1  4998.7  269.43
  5001.5  268.93  5004.7  269.43  5008.3   274.1  5018.6  274.78  5059.7  273.49
  5086.3  275.17  5203.5  274.69  5283.7   277.9  5337.1  280.93  5398.8  286.84
  5831.4  292.22  5891.5  292.57  6181.2  293.79  6433.7  292.47  6507.4  292.82
#Mann= 11 ,-1 , 0
  3950.1     .05       0  3951.1      .1       0  4594.5     .08       0
  4698.6      .1       0  4913.1     .12       0  4998.7     .07       0
  5004.7     .12       0  5283.7     .05       0  5831.4      .1       0
  5891.5     .05       0  6433.7      .1       0
Bank Sta=4975.57,5337.1
XS Rating Curve= 0 ,0
Exp/Cntr=0.3,0.1

Type RM Length L Ch R = 1 ,120812  ,1469,1469,1469
BEGIN DESCRIPTION:
SULPHUR CREEK 121.0
END DESCRIPTION:
XS GIS Cut Line= 3
      2272640.28     13417383.29       2272683.7       13417557.
      2273504.45     13419322.38
#Sta/Elev= 30
  4651.1  290.69  4863.1  291.42  4894.8  289.21  4905.8  287.05  4940.3  281.61
  4946.1  278.73  4962.3  277.54    4969  274.74  4984.4  273.41  4991.9     270
  5003.4  269.38  5006.2  268.88  5009.4  269.38  5014.8  272.91  5058.5  272.75
  5082.5  272.34  5105.7  269.92  5117.4  271.94  5149.8  272.63  5171.9  274.67
  5193.9  278.24  5231.8  283.22  5260.2  284.25  5315.2  282.67  5436.5  282.69
  5524.8  287.85  5586.1  286.54  5648.2  287.76  6277.5  289.43    6777  292.76
#Mann= 7 ,-1 , 0
  4651.1     .05       0  4905.8      .1       0  5003.4     .07       0
  5009.4      .1       0  5058.5     .12       0  5082.5      .1       0
  5648.2     .05       0
Bank Sta=4946.1,5193.9
XS Rating Curve= 0 ,0
Exp/Cntr=0.3,0.1

Type RM Length L Ch R = 1 ,119343  ,474,474,474
BEGIN DESCRIPTION:
SULPHUR CREEK 120.0
END DESCRIPTION:
XS GIS Cut Line= 3
      2272137.73     13417946.81      2271937.72     13418696.85
      2272737.76     13418996.87
#Sta/Elev= 30
  4232.8  289.51  4269.1  289.13  4690.6   287.1  4781.4  285.12  4836.4  277.71
  4871.3  273.15    4978  268.93  4986.4  262.52  4991.6  265.27  4995.7  262.37
  4998.5  261.87  5001.7  262.37  5006.5  265.51  5024.2  268.73  5049.1  266.92
  5054.4  269.31  5079.4  263.82  5104.3  264.73  5109.6  269.02  5134.5  263.97
  5139.9  267.09  5158.6  270.95  5164.8  269.88  5170.1  276.24  5195.1  277.44
    5220  277.01  5297.4  285.13  5457.6  284.85  5817.4   289.8  5863.5   290.7
#Mann= 6 ,-1 , 0
  4232.8      .1       0  4269.1     .05       0  4690.6      .1       0
  4995.7     .07       0  5001.7      .1       0  5817.4     .05       0
Bank Sta=4836.4,5195.1
XS Rating Curve= 0 ,0
Exp/Cntr=0.3,0.1

Type RM Length L Ch R = 1 ,118869  ,1251,1251,1251
BEGIN DESCRIPTION:
SULPHUR CREEK 119.0
END DESCRIPTION:
XS GIS Cut Line= 3
      2271756.41     13417711.23      2271419.56      13418928.3
      2271354.15     13419942.17
#Sta/Elev= 30
  4006.7  287.42  4157.8  287.72  4220.1  285.84  4319.5  287.49  4640.5  285.09
  4666.2     285  4718.1  281.26  4738.8  282.16  4772.7  280.67  4812.2   276.6
    4853   273.2  4904.9  271.57  4967.1  267.43  4977.5  267.97  4996.3  262.24
  4999.1  261.74  5002.3  262.24  5028.5   269.1  5060.5  270.98  5091.6   276.3
  5112.6  280.27  5174.6  287.16  5398.3  282.84  5538.6  284.18  5690.2  283.87
  5736.8  282.39    5843  281.94  5953.4  284.78  6119.8  285.34  6285.5  287.78
#Mann= 6 ,-1 , 0
  4006.7     .05       0  4640.5      .1       0  4996.3     .07       0
  5002.3      .1       0  5736.8     .12       0  5953.4      .1       0
#XS Ineff= 2 , 0
                         5173.97          287.29
Permanent Ineff=
       T       T
Bank Sta=4812.2,5091.6
XS Rating Curve= 0 ,0
Exp/Cntr=0.3,0.1

Type RM Length L Ch R = 1 ,117618  ,1479,1479,1479
BEGIN DESCRIPTION:
Mapping XS 772b3f79
END DESCRIPTION:
XS GIS Cut Line= 3
      2270653.34     13417531.51       2270202.6     13418648.73
      2270384.89     13419785.89
#Sta/Elev= 30
  4070.8  287.72  4077.2  290.43  4101.4  287.72  4119.7  289.29  4152.6  283.29
  4195.2  281.22  4846.3  282.31  4885.3  280.43  4901.2  277.13  4906.9  278.94
  4917.6  274.67  4930.8  274.15  4949.5  269.86  4954.9  272.63  4960.8  267.23
  4984.5   265.1  4993.1  260.26    5003  259.09  5014.7  265.71  5032.8  264.02
  5091.8  266.39  5133.3  273.73  5145.5  278.09  5164.3   276.8  5169.7  279.81
  5223.4  282.29  5374.9  278.24  5406.5  280.61  5783.4  279.16  6427.2  284.63
#Mann= 5 ,-1 , 0
  4070.8     .08       0  4152.6      .1       0  4846.3     .12       0
  4917.6     .07       0  5133.3      .1       0
Bank Sta=4930.8,5133.3
XS Rating Curve= 0 ,0
Exp/Cntr=0.3,0.1

Type RM Length L Ch R = 1 ,116204  ,943,943,943
BEGIN DESCRIPTION:
Mapping XS 31fbf3b0
END DESCRIPTION:
XS GIS Cut Line= 2
      2269318.07     13417631.42      2269268.37     13418543.36
#Sta/Elev= 30
    4904  280.01  4904.1  280.01  4919.5  280.06  4929.5  279.14  4939.5  273.74
  4959.5  270.29  4969.5  269.12  4989.6     264    4997  256.69  4999.8  256.19
  5003.5  257.28  5009.6  256.69  5019.6  258.67  5029.6  262.92  5059.7  263.19
  5099.7  265.48  5119.8  265.75  5129.8   266.7  5139.8  269.01  5149.8  272.83
  5170.6   272.6  5179.8  272.84  5185.5  274.61  5219.9  275.19  5239.9  278.56
    5270   280.2  5650.5  280.04  5690.6   280.6  5730.7  279.56  5817.3  280.54
#Mann= 5 ,-1 , 0
    4904      .1       0  4904.1     .12       0  4959.5     .07       0
  5139.8     .12       0  5170.6      .1       0
Bank Sta=4959.5,5139.8
XS Rating Curve= 0 ,0
Exp/Cntr=0.3,0.1

Type RM Length L Ch R = 1 ,115700  ,885,885,885
BEGIN DESCRIPTION:
Mapping XS 427dbb17
END DESCRIPTION:
XS GIS Cut Line= 3
      2268862.81     13417328.49      2268806.67     13417933.59
      2269006.28     13418457.56
#Sta/Elev= 30
  4443.7  277.53  4557.7  276.76  4673.7  277.65  4693.6  276.11  4705.3  278.33
  4730.6  276.58  4788.7  268.77  4820.3   266.3  4825.6  267.64  4831.6  265.39
  4882.7  262.49  4972.6  262.77    4982   255.9  4992.4  254.86  4995.6  255.36
  5002.7  261.85  5012.7  262.75  5022.8  267.52  5032.8  270.47  5042.9  277.84
  5062.9  279.06  5281.3  278.88  5356.2  272.99  5457.9  275.84  5463.3  277.77
  5482.7  276.48    5506  279.25  5542.9  278.11  5559.5  279.53  5720.8  280.98
#Mann= 5 ,-1 , 0
  4443.7      .1       0  4557.7      .1       0  4693.6     .12       0
  4825.6     .07       0  5032.8      .1       0
#XS Ineff= 2 , 0
                         5118.81          278.79
Permanent Ineff=
       T       T
Bank Sta=4825.6,5022.8
XS Rating Curve= 0 ,0
Exp/Cntr=0.3,0.1

Type RM Length L Ch R = 1 ,114815  ,673,673,673
BEGIN DESCRIPTION:
Mapping XS e6daa8ad
END DESCRIPTION:
XS GIS Cut Line= 2
      2268806.68     13417141.36      2267914.66      13417247.4
#Sta/Elev= 30
  4428.7  276.61    4478  276.06  4548.5  276.46  4568.6  276.01  4598.1  274.36
  4603.1  274.84  4664.9  272.63  4690.8  271.53  4739.8  267.57  4773.4  265.36
  4830.5  261.73  4850.6  261.22    4901  261.71  4951.3  260.37  4961.4  261.37
  4971.5  261.47  4991.6  260.64  5001.7   257.9  5011.5  256.32  5014.7  256.82
  5021.3  258.06  5026.4  258.16  5031.9  262.88 5033.52  265.92 5034.66   267.7
  5041.9  276.17  5072.2  276.89    5114  275.75  5273.6  275.03    5327   275.3
#Mann= 4 ,-1 , 0
  4428.7     .05       0  4664.9      .1       0  4739.8     .07       0
  5014.7      .1       0
Bank Sta=4773.4,5033.52
XS Rating Curve= 0 ,0
Exp/Cntr=0.3,0.1

Type RM Length L Ch R = 1 ,114142  ,665,665,665
BEGIN DESCRIPTION:
SULPHUR CREEK 118.0
END DESCRIPTION:
XS GIS Cut Line= 2
      2268607.09     13416554.97      2267927.15     13416617.35
#Sta/Elev= 30
  4788.5   275.2    4808  275.32  4838.1  276.64  4858.2  276.99  4868.5  276.52
  4888.3  274.67  4908.4  270.58  4918.4  269.29  4928.5  267.09  4938.5  265.91
  4948.5   263.1  4958.6  261.91  4968.4  259.77  4998.7  258.81  5038.9  259.22
  5048.7  258.24    5069  259.94  5099.2  260.95  5109.2  262.05  5119.3  264.08
  5129.3  265.09  5139.3  267.23  5149.4  268.15  5159.4  269.86  5180.6  271.91
  5188.4  272.52  5193.4  271.87  5199.6  273.83  5219.7  275.55  5471.3  274.86
#Mann= 4 ,-1 , 0
  4788.5     .05       0  4938.5     .03       0  5139.3      .1       0
  5180.6     .05       0
Bank Sta=4948.5,5119.3
XS Rating Curve= 0 ,0
Exp/Cntr=0.3,0.1

Type RM Length L Ch R = 1 ,113477  ,792,792,792
BEGIN DESCRIPTION:
SULPHUR CREEK 117.0
END DESCRIPTION:
XS GIS Cut Line= 3
      2268257.74     13415806.38      2267821.05     13416317.93
      2267721.96     13416528.49
#Sta/Elev= 30
  4639.1  273.68  4738.8  273.88  4788.2  273.12  4795.9  271.75  4816.7   270.5
  4823.8  268.82    4831  268.16  4837.6  268.53  4845.3  266.92  4851.9  267.49
  4859.6  266.78  4866.1  266.95  4873.8  265.23  4880.4  265.33  4902.4  262.89
  4915.8  262.25  4923.2  260.52  4951.8  257.79  4980.3   257.5  4986.7  256.78
  5015.5  257.99  5036.3  257.64  5058.3  259.42  5107.7   260.6    5122  262.46
  5136.2  263.02  5206.5  269.73    5235  271.57  5292.1  274.05  5544.4  273.86
#Mann= 3 , 0 , 0
  4639.1     .05       0  4902.4     .03       0  5136.2     .05       0
Bank Sta=4902.4,5136.2
XS Rating Curve= 0 ,0
Exp/Cntr=0.3,0.1

Type RM Length L Ch R = 1 ,112685  ,1055,1055,1055
BEGIN DESCRIPTION:
Mapping XS 7cda2033
END DESCRIPTION:
XS GIS Cut Line= 4
      2267652.65     13415581.81        2267191.     13415931.17
      2266773.05     13416193.17      2266036.97     13416124.55
#Sta/Elev= 30
  4572.9  272.61  4793.5  273.27  4851.7  268.48    4858   266.3  4887.1  261.77
  4894.3  258.44  4943.3  254.86  5027.6  255.65  5107.7  261.77  5136.8  262.52
  5150.8  260.93  5172.7  260.85  5193.9  258.29  5202.9  255.83  5235.3  254.57
  5238.1  254.07  5241.3  254.57  5288.2  256.74  5355.3  263.32    5419  265.25
  5434.3  267.61  5543.9  271.74  5766.5  277.17  5801.1  276.91  5961.8  282.91
  6182.8  288.59  6197.9  290.17  6222.9  288.62    6243  290.14  6384.4  293.68
#Mann= 5 ,-1 , 0
  4572.9     .05       0  4894.3      .1       0  5027.6     .05       0
  5235.3     .07       0  5241.3     .05       0
#XS Ineff= 2 , 0
                         5142.15          262.46
Permanent Ineff=
       T       T
Bank Sta=4887.1,5107.7
XS Rating Curve= 0 ,0
Exp/Cntr=0.3,0.1

Type RM Length L Ch R = 1 ,111630  ,787,787,787
BEGIN DESCRIPTION:
SULPHUR CREEK 116.0
END DESCRIPTION:
XS GIS Cut Line= 3
      2267914.58     13415244.96      2267546.57     13415082.79
      2266112.25     13415064.08
#Sta/Elev= 30
  3799.3  271.82  4240.3  271.23  4460.3  269.96  4530.3  268.49  4590.3  265.99
  4670.3  265.93  4740.4   263.4  4770.4  260.68  4820.4  257.93  4830.4  255.89
  4850.4  254.92  4890.4  255.37  4910.4  254.12  4997.4  252.84  5000.1  252.34
  5003.4  252.84  5010.4  252.94  5100.4  260.54  5140.4  263.24  5170.4  266.26
  5220.4  268.54  5290.4  275.82  5310.4  276.97  5380.4  277.71  5450.4  279.59
  5500.4  282.03  5550.4  283.12  5570.4  282.67  5590.4  283.85  5635.9  284.61
#Mann= 3 ,-1 , 0
  3799.3     .05       0  4997.4     .03       0  5003.4     .05       0
Bank Sta=4770.4,5100.4
XS Rating Curve= 0 ,0
Exp/Cntr=0.3,0.1

Type RM Length L Ch R = 1 ,110843  ,774,774,774
BEGIN DESCRIPTION:
SULPHUR CREEK 115.0
END DESCRIPTION:
XS GIS Cut Line= 3
      2268457.35     13414933.08       2268058.1     13414733.45
       2266482.9     13414191.78
#Sta/Elev= 30
    3535  271.72  3874.4  270.96  4049.1  269.61  4111.6  268.21    4151  266.11
  4262.5  268.83  4267.8  267.95  4293.8  268.35    4373     266    4450  268.95
  4626.8     268  4694.6  267.16  4774.9  260.23  4803.1  257.15  4870.7  253.81
  4954.6  252.53  4975.8  249.23  4998.7  247.99  5001.4  247.49  5004.7  247.99
  5007.5  249.19  5064.1  260.24  5081.5  264.45  5095.4  265.64  5102.7   267.7
  5166.1  274.52  5240.2  275.15  5277.5   276.5  5537.3  278.29  5647.1  278.92
#Mann= 6 ,-1 , 0
    3535     .05       0  4803.1      .1       0  4870.7     .05       0
  4998.7     .03       0  5004.7     .05       0  5537.3      .1       0
Bank Sta=4774.9,5064.1
XS Rating Curve= 0 ,0
Exp/Cntr=0.3,0.1

Type RM Length L Ch R = 1 ,110069  ,641,641,641
BEGIN DESCRIPTION:
SULPHUR CREEK 114.0
END DESCRIPTION:
XS GIS Cut Line= 3
      2268359.97       13414409.      2268157.65     13414157.83
      2267243.78     13413676.48
#Sta/Elev= 30
  4097.9   270.9  4376.9  270.47  4583.8  267.88  4612.5  265.49    4694  263.59
  4710.4  260.84  4754.4   258.2  4820.5  258.16  4858.9  260.93  4886.6  258.02
  4930.7  251.73  4953.4   250.3  4985.5   249.2  4993.8  241.15  4996.5  240.65
  4999.8  241.15  5007.5  241.91  5013.2  248.92  5019.4  250.52  5079.3  252.52
  5095.6  258.68  5101.3  265.24  5109.8  266.36  5123.3  266.63  5139.7  262.37
  5145.3   266.9    5155  262.29  5177.6   267.4  5190.4  267.47  5453.3  270.98
#Mann= 6 ,-1 , 0
  4097.9      .1       0  4376.9     .05       0  4953.4     .12       0
  4993.8     .07       0  4999.8     .12       0  5190.4      .1       0
Bank Sta=4886.6,5095.6
XS Rating Curve= 0 ,0
Exp/Cntr=0.3,0.1

Type RM Length L Ch R = 1 ,109428  ,551,551,551
BEGIN DESCRIPTION:
SULPHUR CREEK 113.0
END DESCRIPTION:
XS GIS Cut Line= 3
      2268722.72     13413502.07      2268332.05     13413390.45
      2267272.22     13413313.75
#Sta/Elev= 30
  4254.6  268.99  4675.3  270.43  4835.7   268.4  4865.8  266.63  4898.5  262.48
  4925.9  257.57  4976.1  249.82  4986.1  240.99  4993.1  239.24  4995.9  238.74
  4999.1  239.24  5006.1  244.83  5016.2  248.27  5026.2  246.38  5046.2  249.47
  5076.3  249.73  5186.6  257.48  5193.6  258.85  5198.6  257.28  5206.7  257.68
  5224.3  261.11  5246.8  260.28  5286.9  263.26  5306.9  266.69    5327  267.32
  5408.9  266.62  5472.5  264.75  5512.6  266.72  5577.6  269.04  5723.5   269.8
#Mann= 7 ,-1 , 0
  4254.6     .05       0  4898.5      .1       0  4993.1     .07       0
  4999.1      .1       0  5224.3      .1       0  5408.9     .12       0
  5512.6      .1       0
Bank Sta=4925.9,5186.6
XS Rating Curve= 0 ,0
Exp/Cntr=0.3,0.1

Type RM Length L Ch R = 1 ,108877  ,854,854,854
BEGIN DESCRIPTION:
SULPHUR CREEK 112.0
END DESCRIPTION:
XS GIS Cut Line= 3
      2269343.55     13412895.14      2268555.29     13412874.21
      2267634.42     13412825.38
#Sta/Elev= 30
  3799.8  269.56  3975.7  267.36  4125.7   261.9  4255.8  267.13  4275.8  266.31
  4455.9  267.96  4816.2  268.09  4886.3  267.16  4935.4  263.45  4956.4  259.07
  4966.4  255.19  4986.5  240.48  4993.5  239.81  4996.2  239.31  4999.5  239.81
    5006  243.11    5011  241.29  5016.5  245.49  5026.5  249.48  5062.6  247.64
  5096.6  249.96  5136.7     249  5166.7  250.17  5226.8  253.62  5246.8  256.55
  5256.8  256.34  5280.1  260.29  5326.9  265.43    5367  266.78  5510.5  266.74
#Mann= 6 ,-1 , 0
  3799.8     .05       0  4935.4      .1       0  4993.5     .07       0
  4999.5      .1       0  5062.6     .12       0  5280.1      .1       0
#XS Ineff= 2 , 0
         4454.55  267.98
Permanent Ineff=
       T       T
Bank Sta=4966.4,5246.8
XS Rating Curve= 0 ,0
Exp/Cntr=0.3,0.1

Type RM Length L Ch R = 1 ,108023  ,692,692,692
BEGIN DESCRIPTION:
SULPHUR CREEK 111.0
END DESCRIPTION:
XS GIS Cut Line= 3
      2269176.19     13412406.83      2269057.57     13412295.19
        2268046.     13412071.95
#Sta/Elev= 30
  4184.1  267.16    4394  266.33  4493.9  264.29  4613.1  260.33  4633.6  254.76
  4639.8  259.72  4761.8  264.69    4776  264.45  4781.1   261.3  4797.4  259.52
  4824.8  261.65  4856.9  258.95  4868.4  257.91  4873.6  254.15  4889.6  254.37
  4930.6  248.37  4971.5  247.78  4981.8   245.6    4992  238.32  4999.2  237.24
    5002  236.74  5005.2  237.24  5014.9  244.92  5022.7  247.32  5094.4  248.67
  5114.9  255.02  5135.4  258.14  5157.5  264.35  5227.5     267  5382.9  266.62
#Mann= 8 ,-1 , 0
  4184.1     .05       0    4394      .1       0  4493.9     .12       0
  4761.8      .1       0  4856.9     .12       0  4999.2     .07       0
  5005.2     .12       0  5157.5      .1       0
#XS Ineff= 2 , 0
         4765.23  265.01
Permanent Ineff=
       T       T
Bank Sta=4889.6,5114.9
XS Rating Curve= 0 ,0
Exp/Cntr=0.3,0.1

Type RM Length L Ch R = 1 ,107331  ,675,675,675
BEGIN DESCRIPTION:
SULPHUR CREEK 110.0
END DESCRIPTION:
XS GIS Cut Line= 3
       2269413.4      13411681.3      2269183.15     13411597.57
      2268262.47     13411492.95
#Sta/Elev= 30
  4146.9  266.04  4444.9  264.74  4508.1   263.9  4518.1  261.03  4538.3  258.62
  4568.5  259.55  4578.5  255.68  4588.6     256  4618.2  251.33  4628.8  248.62
  4638.9  249.79  4669.1  257.39  4706.6  260.35  4759.7  262.36  4800.9  256.28
  4840.2  254.41  4859.7  250.08  4950.9  245.41    4975  245.93  4981.1  245.32
  4998.2  236.99    5001  236.49  5004.2  236.99  5021.4  246.89  5031.4  245.84
  5048.3  247.32  5111.9  254.54  5172.3  263.41  5238.7  265.11  5318.5  264.75
#Mann= 8 ,-1 , 0
  4146.9     .05       0  4444.9     .16       0  4618.2     .12       0
  4706.6     .16       0  4859.7     .12       0  4998.2     .07       0
  5004.2     .12       0  5048.3      .1       0
#XS Ineff= 2 , 0
         4758.86  262.55
Permanent Ineff=
       T       T
Bank Sta=4840.2,5111.9
XS Rating Curve= 0 ,0
Exp/Cntr=0.3,0.1

Type RM Length L Ch R = 1 ,106656  ,571,571,571
BEGIN DESCRIPTION:
SULPHUR CREEK 109.0
END DESCRIPTION:
XS GIS Cut Line= 3
      2269559.86      13411297.6      2269287.79     13411074.36
      2268415.78     13410774.38
#Sta/Elev= 30
  4078.2  265.46  4308.1  264.61  4475.9   264.3  4561.6  260.48  4578.3  263.98
  4621.4  262.96  4705.2  256.82  4712.5  251.92    4758  246.92  4774.9  242.08
  4800.3  249.22  4806.2   254.3  4837.4  257.69 4855.91  253.84  4874.4  245.66
  4884.9  244.73  4948.4  245.14  4962.3  242.11  4980.1   245.1  4988.3  236.79
  4998.3  236.14    5001  235.64  5004.3  236.14  5011.8  245.39    5082  251.29
  5131.2  252.34  5144.5  253.93  5149.7  257.21  5191.6  262.04  5352.3  263.91
#Mann= 7 ,-1 , 0
  4078.2      .1       0  4308.1     .05       0  4475.9      .1       0
  4621.4     .12       0  4998.3     .07       0  5004.3     .12       0
  5131.2      .1       0
#XS Ineff= 2 , 0
         4838.41  257.69
Permanent Ineff=
       T       T
Bank Sta=4855.91,5144.5
XS Rating Curve= 0 ,0
Exp/Cntr=0.3,0.1

Type RM Length L Ch R = 1 ,106085  ,643,643,643
BEGIN DESCRIPTION:
SULPHUR CREEK 108.0
END DESCRIPTION:
XS GIS Cut Line= 3
      2269748.24     13411123.22      2269392.43     13410467.43
      2268534.38      13410272.1
#Sta/Elev= 30
  3827.8  265.46    4106  263.45  4262.5  263.28  4303.9  264.41  4429.4  264.38
  4467.5  263.46  4763.3  262.24  4835.1  256.96  4845.4  257.15  4870.2  253.39
  4876.2  251.25  4886.4   250.3  4896.1  247.54  4913.2  245.13  4968.5  243.96
  4978.7  241.49    4989  237.28  4996.2  236.07    4999  235.57  5002.2  236.07
  5004.4  242.59  5009.5  244.29  5040.2     244  5081.3  248.28 5097.84  253.05
    5112  258.04  5157.4  262.28  5321.1  260.97    5430   264.1  5453.9   263.8
#Mann= 7 ,-1 , 0
  3827.8      .1       0    4106     .05       0  4262.5      .1       0
  4896.1     .12       0  4996.2     .07       0  5002.2     .12       0
  5157.4      .1       0
#XS Ineff= 2 , 0
                            5157          262.59
Permanent Ineff=
       T       T
Bank Sta=4870.2,5097.84
XS Rating Curve= 0 ,0
Exp/Cntr=0.3,0.1

Type RM Length L Ch R = 1 ,105442  ,782,782,782
BEGIN DESCRIPTION:
SULPHUR CREEK 107.0
END DESCRIPTION:
XS GIS Cut Line= 3
      2270194.69     13409783.76      2268820.38     13409762.83
      2268373.91      13409860.5
#Sta/Elev= 30
  3982.5  273.37  4030.1  272.82  4206.9  267.09  4369.9  260.85  4429.5  260.06
  4489.5  253.67  4729.6     247  4759.5  249.47  4764.5  247.92  4809.6  254.08
  4849.6     255  4879.6  251.68    4888  250.15  4949.6  242.64  4969.6  243.13
  4986.6  236.04  4989.3  235.54  4992.6  236.04  5019.6  244.26  5089.6  245.49
  5109.6  247.96  5119.6  251.81  5182.4  260.26  5199.6  261.72  5219.6  259.47
  5229.6  261.78  5279.6  263.04    5503  260.01  5646.3  263.18    5814   263.2
#Mann= 8 ,-1 , 0
  3982.5      .1       0  4030.1     .05       0  4206.9      .1       0
  4369.9     .05       0    4888     .12       0  4986.6     .07       0
  4992.6     .12       0  5182.4      .1       0
#XS Ineff= 2 , 0
         4849.43  255.03 5349.36          263.49
Permanent Ineff=
       T       T
Bank Sta=4879.6,5119.6
XS Rating Curve= 0 ,0
Exp/Cntr=0.3,0.1

Type RM Length L Ch R = 1 ,104660  ,669,669,669
BEGIN DESCRIPTION:
SULPHUR CREEK 106.0
END DESCRIPTION:
XS GIS Cut Line= 4
      2269811.02     13408667.55      2269538.93     13408904.76
      2268562.26     13409232.64      2267948.34     13409609.37
#Sta/Elev= 30
    4333   275.9  4384.5  273.17  4705.8  264.72  4769.1  262.08  4795.6  258.14
    4864  254.95  4895.7  251.03  4934.4  244.76  4939.7  246.06    4959  241.98
  4976.7  243.46  4990.6  240.58  4994.5  236.38  4997.2  235.88  5000.5  236.38
  5022.3  242.58  5060.5  242.17  5092.1  244.37  5180.5  243.47  5264.9  250.71
  5306.4     254  5328.2  256.28  5454.7  256.57  5475.8  259.76  5496.7  260.73
  5722.7  263.21  5854.6  262.67  6022.8  257.85  6239.4  262.52  6444.5  260.88
#Mann= 6 ,-1 , 0
    4333      .1       0  4795.6     .05       0  4976.7     .12       0
  4994.5     .07       0  5000.5     .12       0  5306.4      .1       0
#XS Ineff= 2 , 0
                         5775.11          263.18
Permanent Ineff=
       T       T
Bank Sta=4895.7,5264.9
XS Rating Curve= 0 ,0
Exp/Cntr=0.3,0.1

Type RM Length L Ch R = 1 ,103991  ,592,592,592
BEGIN DESCRIPTION:
SULPHUR CREEK 105.0
END DESCRIPTION:
XS GIS Cut Line= 4
      2269748.24     13408367.59      2269259.88     13408374.57
      2268352.98     13408611.76      2267746.28     13409302.14
#Sta/Elev= 30
  4107.4  276.98  4583.4  262.46  4664.7  260.92  4705.1   257.5  4781.8  255.66
  4826.4   254.6  4877.1  248.95  4896.9  245.89  4959.8  240.79    4983   241.8
  4990.8  240.19  4998.2  234.49  5000.9  233.99  5004.2  234.49  5011.5   234.7
  5018.2  239.15  5023.4  240.21  5117.4  246.24  5139.5  250.32  5215.2  258.69
  5238.9  255.54  5296.1  259.84  5321.6  257.32  5331.4  259.47  5342.3  259.83
  5915.9  261.52    5987  260.75  6128.4  255.76  6263.1  261.59  6452.3  260.46
#Mann= 6 ,-1 , 0
  4107.4      .1       0  4583.4     .05       0  4781.8     .12       0
  4998.2     .07       0  5004.2     .12       0  5117.4      .1       0
#XS Ineff= 2 , 0
                         5821.08          261.93
Permanent Ineff=
       T       T
Bank Sta=4877.1,5139.5
XS Rating Curve= 0 ,0
Exp/Cntr=0.3,0.1

Type RM Length L Ch R = 1 ,103399  ,696,696,696
BEGIN DESCRIPTION:
SULPHUR CREEK 104.0
END DESCRIPTION:
XS GIS Cut Line= 3
      2269343.61     13407579.27       2269078.5     13407823.45
      2267872.87      13408171.9
#Sta/Elev= 30
  4196.1  281.58  4283.7  278.91  4396.5  272.17  4418.1  272.95  4481.6   267.2
  4519.1  266.26    4535  265.48  4671.9  258.92  4735.2  252.54  4775.9  243.36
  4796.8  242.77    4828  247.11  4848.8  242.23  4869.6  241.28  4963.3  243.06
  4986.1   239.1  4994.5  234.37  5001.9  233.47  5004.7  232.97  5007.9  233.47
  5038.3  241.89  5046.6  243.08  5053.4  246.74  5058.6  249.91  5077.8   250.8
    5109  259.03  5421.3  257.99  5535.8   253.2  5666.6  258.07  5811.5  258.54
#Mann= 7 ,-1 , 0
  4196.1     .05       0  4519.1     .16       0    4535     .05       0
  4671.9     .12       0  5001.9     .07       0  5007.9     .12       0
  5038.3      .1       0
#XS Ineff= 2 , 0
                         5154.17          259.53
Permanent Ineff=
       T       T
Bank Sta=4828,5053.4
XS Rating Curve= 0 ,0
Exp/Cntr=0.3,0.1

Type RM Length L Ch R = 1 ,102703  ,773,773,773
BEGIN DESCRIPTION:
SULPHUR CREEK 103.0
END DESCRIPTION:
XS GIS Cut Line= 4
      2269455.21      13407223.5      2269022.69     13407139.79
      2268192.53     13407404.88      2267746.01       13407670.
#Sta/Elev= 30
  4085.8  285.49  4236.3  280.12  4511.3  269.09  4594.1  265.95  4599.4  255.08
    4605  261.11  4615.5  261.29  4636.8  249.68  4695.9  248.77    4710  255.44
  4728.1  251.45  4733.3  255.23    4773  249.72  4804.5   256.1    4815  255.68
  4824.6  247.63    4836  246.41  4838.3  246.26  4990.8  238.91    5001  233.28
  5003.7  232.78    5007  233.28    5023  239.57  5092.6  241.73  5116.2  245.69
  5140.4  247.14  5162.2  252.02  5339.9  257.77  5564.3  250.99  5917.1  257.78
#Mann= 7 ,-1 , 0
  4085.8     .05       0  4236.3      .1       0  4511.3     .05       0
  4838.3     .12       0    5001     .07       0    5007     .12       0
  5116.2      .1       0
#XS Ineff= 1 ,-1
 5357.85 5900.99  258.04
Permanent Ineff=
       T
Bank Sta=4836,5140.4
XS Rating Curve= 0 ,0
Exp/Cntr=0.3,0.1

Type RM Length L Ch R = 1 ,101930  ,1089,1089,1089
BEGIN DESCRIPTION:
SULPHUR CREEK 102.0
END DESCRIPTION:
XS GIS Cut Line= 4
      2269224.96     13406672.37      2268590.17     13406463.09
      2266818.22     13407160.71      2266253.58     13407732.33
#Sta/Elev= 30
    3944  273.38  4358.9  259.68  4845.5  256.64  4909.9  255.88  4915.9  252.23
  4934.3  250.45  4939.7  245.84  4980.4   238.4  4990.9  232.38  4993.6  231.88
  4996.9  232.38  5066.4  241.79    5132  239.72  5277.8  246.32  5289.1  246.92
  5421.1   254.8  5511.1  249.18  5517.8  244.89  5535.5  241.85  5582.3  242.41
  5657.5   250.3    5679  259.28    5698  260.34  5733.2  252.65  5797.2  248.87
  5979.9  244.26  6196.3   248.7    6245  256.42  6832.6   255.3  7320.2  261.22
#Mann= 5 ,-1 , 0
    3944      .1       0  4845.5     .12       0  4990.9     .07       0
  4996.9     .12       0  5277.8      .1       0
#XS Ineff= 2 ,-1
 5417.96 5661.24  254.61 5689.53 7279.35  260.37
Permanent Ineff=
       T       T
Bank Sta=4939.7,5289.1
XS Rating Curve= 0 ,0
Exp/Cntr=0.3,0.1

Type RM Length L Ch R = 1 ,100841  ,420,420,420
BEGIN DESCRIPTION:
SULPHUR CREEK 101.0
END DESCRIPTION:
XS GIS Cut Line= 3
       2268453.7      13405502.8      2267341.87     13406010.04
      2266189.04     13407065.51
#Sta/Elev= 30
  3777.9   257.9  4472.9  254.59  4487.9  253.78  4501.4  249.44  4547.5  245.97
  4577.1  251.59  4719.7  245.09  4949.6   239.1  4984.2   236.2  4996.5  231.61
  4999.3  231.11  5002.5  231.61  5035.9  245.14  5044.1  246.65  5064.3  245.13
    5100  237.82  5135.2  237.19  5163.5  237.68  5234.5  245.78  5397.3  252.08
  5446.6  252.41  5467.5  248.14  5510.1  247.15  5560.1  249.87  5566.8  252.33
  5793.1  255.56  5977.5  254.51  6132.9  250.08  6168.7  253.05    6563   257.4
#Mann= 5 ,-1 , 0
  3777.9      .1       0  4577.1     .12       0  4996.5     .07       0
  5002.5     .12       0  5044.1      .1       0
#XS Ineff= 2 , 0
                         5832.67          255.83
Permanent Ineff=
       T       T
Bank Sta=4719.7,5035.9
XS Rating Curve= 0 ,0
Exp/Cntr=0.3,0.1

Type RM Length L Ch R = 1 ,100421  ,1063,1063,1063
BEGIN DESCRIPTION:
SULPHUR CREEK 100.0
END DESCRIPTION:
XS GIS Cut Line= 3
      2269787.71     13404796.86      2267087.72     13405696.85
      2265087.77     13406096.85
#Sta/Elev= 30
  2128.9  281.94  2782.4  265.22  4152.7  252.77  4532.2  255.09  4637.6  253.39
  4658.7  248.72  4669.3  251.75    4720  246.04    4743  245.16  4977.5  237.45
  5002.5  231.04  5005.3  230.54  5008.5  231.04  5025.9  237.72  5109.7  239.99
  5270.7   244.7  5372.7  250.85  5586.8  253.15    5750  249.52  5821.4  241.64
  5923.4  248.68  5964.1  246.32  6004.9  251.23  6035.5  246.98  6147.7  247.43
  6188.5  249.58  6208.9  255.35  6361.9  254.94  6423.1  261.08  7014.5  278.21
#Mann= 5 ,-1 , 0
  2128.9      .1       0    4720     .12       0  5002.5     .07       0
  5008.5     .12       0  5109.7      .1       0
#XS Ineff= 2 , 0
            4529  255.05
Permanent Ineff=
       T       T
Bank Sta=4743,5270.7
XS Rating Curve= 0 ,0
Exp/Cntr=0.3,0.1

Type RM Length L Ch R = 1 ,99358   ,845,845,845
BEGIN DESCRIPTION:
SULPHUR CREEK 99.0
END DESCRIPTION:
XS GIS Cut Line= 3
      2268840.24     13404620.45      2267320.71     13404738.35
      2265304.57     13405432.22
#Sta/Elev= 30
  2379.9  262.73  3144.7  251.36  3561.2  252.99    3897  249.64  4225.9  252.66
  4573.4  251.38    4584  249.79  4684.4  247.18  4740.9  245.77  4753.2  242.71
  4763.8  239.93  4784.9  238.42    4859  236.38  4933.6  236.73    4969  234.25
    5004  228.56  5006.8  228.06    5010  228.56    5022   230.5  5028.2  239.38
  5038.8  242.29  5053.2  242.11  5070.5  244.35  5110.4  247.07  5146.9  246.89
  5165.7  249.73  5186.8  248.87  5240.6  253.04  5345.4  256.17  6036.2  270.35
#Mann= 5 ,-1 , 0
  2379.9      .1       0  4684.4     .12       0    4969      .1       0
    5004     .07       0    5010      .1       0
#XS Ineff= 2 , 0
         4214.99  252.71
Permanent Ineff=
       T       T
Bank Sta=4753.2,5070.5
XS Rating Curve= 0 ,0
Exp/Cntr=0.3,0.1

Type RM Length L Ch R = 1 ,98513   ,689,689,689
BEGIN DESCRIPTION:
SULPHUR CREEK 97.0
END DESCRIPTION:
XS GIS Cut Line= 3
      2267792.29      13403965.5      2265408.23     13404437.07
      2265067.63     13404869.36
#Sta/Elev= 30
  3204.4  256.66  3637.2  248.88  3881.8  247.46    4208  251.02  4503.7  250.83
    4676  244.34  4758.3  245.21  4829.8  242.57  4840.1  241.51  4870.6  234.08
  4886.1  232.58  4921.6  232.37  4952.2  235.18  4993.7  230.96  5000.2  227.92
  5002.9  227.42  5006.2  227.92  5013.3  233.08  5023.5  233.56  5039.9  238.63
    5045  236.52  5074.5  240.41  5091.1  240.71 5096.02  242.98  5096.2  239.96
 5103.98  243.35  5115.3  248.22  5135.7  250.97  5193.6  253.39    6185  272.93
#Mann= 4 ,-1 , 0
  3204.4      .1       0  4758.3     .16       0  5000.2     .07       0
  5006.2      .1       0
Bank Sta=4829.8,5103.98
XS Rating Curve= 0 ,0
Exp/Cntr=0.3,0.1

Type RM Length L Ch R = 1 ,97824   ,907,907,907
BEGIN DESCRIPTION:
SULPHUR CREEK 96.0
END DESCRIPTION:
XS GIS Cut Line= 4
        2267491.     13403454.63      2266953.93     13403310.54
      2265054.55      13403939.3      2264832.31     13404344.55
#Sta/Elev= 30
  3372.7  255.89  3552.1  254.81  3862.7  247.49  4033.3  246.78  4179.9  246.67
  4697.1  249.75    4792  250.32  4819.4     246  4841.2  248.83  4901.2  243.21
  4919.8  241.05  4925.5  236.77    4936  236.21  4946.2  231.36  4983.2   231.6
  4996.2  226.19    4999  225.69  5002.2  226.19  5009.7  230.73  5020.3   232.9
  5072.9  233.87    5147  241.29  5173.5  238.48  5188.8  242.25  5270.8  243.95
  5522.3  252.87  5886.6  261.19  6086.8  267.21  6136.7  267.45  6391.7   273.6
#Mann= 12 ,-1 , 0
  3372.7     .05       0  4033.3      .1       0  4179.9     .05       0
  4697.1      .1       0    4792     .16       0  4901.2     .12       0
  4996.2     .07       0  5002.2     .12       0  5270.8      .1       0
  5886.6     .05       0  6086.8      .1       0  6136.7     .05       0
#XS Ineff= 2 , 0
         4787.13  250.65
Permanent Ineff=
       T       T
Bank Sta=4919.8,5147
XS Rating Curve= 0 ,0
Exp/Cntr=0.3,0.1

Type RM Length L Ch R = 1 ,96917   ,971,971,971
BEGIN DESCRIPTION:
Mapping XS 174b8818
END DESCRIPTION:
XS GIS Cut Line= 4
      2267495.37     13403171.76      2266106.52     13402477.34
       2264821.8     13403380.12      2264631.76     13403673.82
#Sta/Elev= 30
  2588.8  252.93  4248.9  244.09    4499  247.86    4813  246.76  4858.8  246.19
  4915.5  239.19  4986.9  230.65  4998.7  226.44  5001.5  225.94  5004.7  226.44
  5007.9  230.06  5123.7  234.38  5144.6   238.8  5146.1  238.68  5195.2  239.94
    5210  244.87    5311  247.42  5325.7  247.42    5332  243.26  5361.6  243.37
  5367.7  248.43  5382.5  242.91  5397.3  243.18  5403.4  246.96  5418.2  243.05
  5468.8  243.71  5504.5   245.3  5546.3  253.66  6020.8  266.22  6061.6  267.08
#Mann= 6 ,-1 , 0
  2588.8     .05       0    4813     .12       0  4998.7     .07       0
  5004.7     .12       0  5146.1      .1       0  6020.8     .05       0
#XS Ineff= 2 , 0
         4720.45  248.41
Permanent Ineff=
       T       T
Bank Sta=4915.5,5144.6
XS Rating Curve= 0 ,0
Exp/Cntr=0.3,0.1

Type RM Length L Ch R = 1 ,95946   ,1409,1409,1409
BEGIN DESCRIPTION:
SULPHUR CREEK 95.0
END DESCRIPTION:
XS GIS Cut Line= 4
      2267464.81     13401843.43      2265028.35     13401843.43
      2264360.29     13402904.46      2264216.48     13403793.51
#Sta/Elev= 30
  2068.2  253.17  2104.2  252.87  2677.5  247.21  2965.3  244.95    3153  249.19
  3331.3  250.02  3434.8  247.78  3615.3  242.73  4720.6  245.12  4797.5  245.57
  4812.8  239.71  4818.7  245.19    4834  238.79  4839.9  245.99  4849.3  239.29
  4876.4  236.18  4910.3  235.47  4941.8  234.34  4998.2  224.63  5000.9  224.13
  5004.2  224.63  5022.4   229.9  5117.8  231.58  5231.4  236.28  5241.3  237.15
  5704.1  249.59  5810.2  254.69  6293.7  267.94  6497.7  273.56  6659.1  277.22
#Mann= 17 ,-1 , 0
  2068.2      .1       0  2104.2     .05       0  2677.5      .1       0
    3153     .05       0  3331.3      .1       0  3434.8     .05       0
  4720.6      .1       0  4910.3     .12       0  4941.8      .1       0
  4998.2     .07       0  5004.2      .1       0  5117.8     .12       0
  5231.4      .1       0  5704.1     .05       0  5810.2      .1       0
  6293.7     .05       0  6497.7      .1       0
#XS Ineff= 2 , 0
         4227.27  246.66
Permanent Ineff=
       T       T
Bank Sta=4876.4,5241.3
XS Rating Curve= 0 ,0
Exp/Cntr=0.3,0.1

Type RM Length L Ch R = 1 ,94537   ,1012,1012,1012
BEGIN DESCRIPTION:
Mapping XS 15559947
END DESCRIPTION:
XS GIS Cut Line= 2
      2267634.33     13401522.48      2262877.38     13401157.89
#Sta/Elev= 30
  1464.2  256.44  1843.7  251.21  2059.5  248.41    2504  244.49  2669.9  245.63
    2895  247.91    3226  241.93  3677.3  246.63    4085  245.05  4359.3   238.1
  4463.7  240.66  4529.8  241.35  4630.1   235.7  4744.6  231.22  4879.5   229.9
    4951   227.5    4961  226.81  4971.1  221.95  5002.9  221.81  5005.6  221.31
  5008.9  221.81  5011.2  228.51  5075.2  232.19  5111.5  235.01  5121.5  238.15
  5136.5  238.86  5141.6  243.43  5161.6  250.79  5191.7  252.63  6235.1  266.52
#Mann= 11 ,-1 , 0
  1464.2     .05       0  1843.7      .1       0  2059.5     .05       0
    2504      .1       0  2669.9     .05       0    4085      .1       0
  4463.7     .05       0  4879.5     .12       0  5002.9     .07       0
  5008.9     .12       0  5075.2      .1       0
#XS Ineff= 2 , 0
         3676.14   246.6
Permanent Ineff=
       T       T
Bank Sta=4630.1,5111.5
XS Rating Curve= 0 ,0
Exp/Cntr=0.3,0.1

Type RM Length L Ch R = 1 ,93525   ,403,403,403
BEGIN DESCRIPTION:
SULPHUR CREEK 94.0
END DESCRIPTION:
XS GIS Cut Line= 3
      2267837.71     13400896.85      2264837.72     13400596.85
      2262837.77     13400596.85
#Sta/Elev= 30
  1985.6  262.38  2133.8  261.12  2749.4  248.17  3191.6  244.85  3468.2  245.93
    3709  243.78    3917  240.13  4005.6  237.72  4143.8  243.92    4287  245.01
  4763.7  244.44  4829.7  242.35  4852.3  237.14    4892  234.82  4980.4  224.46
    4995  218.28  4997.8  217.78    5001  218.28  5010.5  223.33  5050.5  226.99
  5160.5  229.01 5176.14  234.11  5180.5  235.78  5247.3   236.9  5270.5  235.36
  5300.5  239.13  5390.5  243.09  5530.5  241.82  6480.5   254.4  7000.5  266.56
#Mann= 9 ,-1 , 0
  1985.6      .1       0  3468.2     .05       0    3709      .1       0
    3917     .05       0  4763.7      .1       0    4892     .12       0
    4995     .07       0    5001     .12       0  5247.3      .1       0
#XS Ineff= 2 , 0
          4289.2  245.07
Permanent Ineff=
       T       T
Bank Sta=4892,5176.14
XS Rating Curve= 0 ,0
Exp/Cntr=0.3,0.1

Type RM Length L Ch R = 1 ,93122   ,698,698,698
BEGIN DESCRIPTION:
SULPHUR CREEK 93.0
END DESCRIPTION:
XS GIS Cut Line= 3
      2266777.61     13400315.52      2264238.53     13400228.72
      2262981.28     13400293.75
#Sta/Elev= 30
    3234  245.53  3514.1  244.01    3923  246.04  4084.4  243.68    4182  239.31
  4249.2  235.86  4464.6  242.86  4806.2  243.27  4854.8  243.71  4878.4  241.35
  4924.9  234.38  4954.9  227.28  4984.9  224.01  4991.9  217.72  4994.7  217.22
  4997.9  217.72  5004.9  218.04  5014.9  224.94    5055  228.47    5175  226.15
    5205  230.21  5255.1  233.24  5305.1  236.65  5345.1  235.62  5404.9  237.48
  5505.2  242.51  5695.3   240.9  5845.5  242.26  6610.6  253.95  7033.5  263.12
#Mann= 8 ,-1 , 0
    3234     .05       0    4182      .1       0  4249.2     .05       0
  4806.2      .1       0  4878.4     .12       0  4991.9     .07       0
  4997.9     .12       0  5404.9      .1       0
#XS Ineff= 2 , 0
         4855.11  244.02
Permanent Ineff=
       T       T
Bank Sta=4924.9,5255.1
XS Rating Curve= 0 ,0
Exp/Cntr=0.3,0.1

Type RM Length L Ch R = 1 ,92424   ,1044,1044,1044
BEGIN DESCRIPTION:
SULPHUR CREEK 92.0
END DESCRIPTION:
XS GIS Cut Line= 4
      2266429.91     13399590.37      2265696.41     13399564.17
      2263587.44     13399655.87       2262696.7     13400035.74
#Sta/Elev= 30
  3435.8  254.08  3505.2  252.67  3628.1  250.59  3840.1  242.38  4035.7  242.58
  4129.1  242.54    4212   242.4  4498.8  240.16  4578.1  236.35    4699  229.88
  4799.1  238.67  4903.7  240.77  4909.2  240.45 4926.14  232.83  4929.2  229.38
  4939.2  227.73  4989.2  223.22  4996.2   216.6    4999   216.1  5002.2   216.6
  5009.3  216.72  5019.3  223.41  5149.4  225.59  5199.4  232.25  5285.7  237.57
  5501.2  239.41  5589.8  237.33  5609.8  234.79    5750   240.4  7249.1  265.44
#Mann= 11 ,-1 , 0
  3435.8      .1       0  3505.2     .05       0  3840.1      .1       0
  4035.7     .05       0  4129.1      .1       0    4212     .05       0
  4578.1      .1       0  4903.7     .12       0  4996.2     .07       0
  5002.2     .12       0  5285.7      .1       0
#XS Ineff= 2 , 0
         4892.05  240.94
Permanent Ineff=
       T       T
Bank Sta=4926.14,5199.4
XS Rating Curve= 0 ,0
Exp/Cntr=0.3,0.1
